--- Rocky Cedar Creek.prj (project) ---

Proj Title=Rocky Cedar Creek Base Level Engineering
Current Plan=p01
Default Exp/Contr=0.3,0.1
English Units
Geom File=g01
Flow File=f01
Plan File=p01
Y Axis Title=Elevation
X Axis Title(PF)=Main Channel Distance
X Axis Title(XS)=Station
BEGIN DESCRIPTION:
Rocky Cedar Creek
END DESCRIPTION:
DSS File=dss
DSS Export Rating Curves= 0
DSS Export Rating Curve Sorted= 0
DSS Export Volume Flow Curves= 0
DXF OffsetX= 0
DXF OffsetY= 0
DXF ScaleX= 1
DXF ScaleY= 10

--- Rocky Cedar Creek.p01 (plan) ---

Plan Title=Multiple Run
Program Version=4.10
Short Identifier=Multiple Run
Geom File=g01
Flow File=f01
Subcritical Flow
K Sum by GR= 0
Std Step Tol= 0.01
Critical Tol= 0.01
Num of Std Step Trials= 20
Max Error Tol= 0.3
Flow Tol Ratio= 0.001
Split Flow NTrial= 30
Split Flow Tol= 0.02
Split Flow Ratio= 0.02
Log Output Level= 0
Friction Slope Method= 1
Unsteady Friction Slope Method= 2
Unsteady Bridges Friction Slope Method= 1
Parabolic Critical Depth
Global Vel Dist= 1 , 1 , 1
Global Log Level= 0
CheckData=True
Encroach Param=-1 ,0,0, 0
BEGIN DESCRIPTION:
Multiple Run
END DESCRIPTION:
Computation Interval=1HOUR
Output Interval=1HOUR
Run HTab= 0
Run UNet= 0
Run PostProcess= 0
Run WQNet= 0
UNET Theta= 1
UNET Theta Warmup= 1
UNET ZTol= 0.02
UNET ZSATol= 0.05
UNET MxIter= 20
UNET MaxInSteps= 0
UNET DtIC= 0
UNET DtMin= 0
UNET MaxCRTS= 20
UNET WFStab= 2
UNET SFStab= 1
UNET WFX= 1
UNET SFX= 1
UNET DSS MLevel= 4
UNET DZMax Abort= 100
UNET Convert EG Bridges= 0
UNET Use Existing IB Tables=-1
UNET Froude Reduction=False
UNET Froude Limit= 1
UNET Froude Power= 10
UNET Time Slicing=0,0, 5
UNET Junction Losses=0
Instantaneous Interval=1HOUR
DSS File=dss
Write IC File= 0
Write IC File at Sim End=0
Echo Input=False
Echo Parameters=False
Echo Output=False
Write Detailed= 0
WQ AD Non Conservative
WQ ULTIMATE=-1
WQ Max Comp Step=1HOUR
WQ Output Interval=15MIN
WQ Output Selected Increments= 0
WQ Output face flow=0
WQ Output face velocity=0
WQ Output face area=0
WQ Output face dispersion=0
WQ Output cell volume=0
WQ Output cell surface area=0
WQ Output cell continuity=0
WQ Output cumulative cell continuity=0
WQ Output face conc=0
WQ Output face dconc_dx=0
WQ Output face courant=0
WQ Output face peclet=0
WQ Output face adv mass=0
WQ Output face disp mass=0
WQ Output cell mass=0
WQ Output cell source sink temp=0
WQ Output cell source sink nsm=0
WQ Output MaxMinRange=-1
WQ Daily Max Min Mean=-1
WQ Daily Range=0
WQ Daily Time=0
WQ Create Restart=0
WQ Fixed Restart=0
WQ System Summary=0
WQ Use Fixed Temperature=0
Sorting and Armoring Iterations= 10
XS Update Threshold= 0.02
Hydraulics Update Threshold= 0.02
Energy Slope Method= 1
Volume Change Method= 0
XS Weighting Method= 0
Number of US Weighted Cross Sections= 1
Number of DS Weighted Cross Sections= 1
Upstream XS Weight=0.25
Main XS Weight=0.5
Downstream XS Weight=0.25
Number of DS XS's Weighted with US Boundary= 1
Upstream Boundary Weight= 1
Weight of XSs Associated with US Boundary= 0
Number of US XS's Weighted with DS Boundary= 1
Downstream Boundary Weight= 0.5
Weight of XSs Associated with DS Boundary= 0.5
Sediment Output Level= 4
Mass or Volume Output= 0
Output Increment Type= 1
Profile and TS Output Increment= 10
XS Output Flag= 0
XS Output Increment= 10
Disregard all LS=0
Disregard all Conn=0
Disregard all Breaches=0
Disregard all Pumps=0

--- Rocky Cedar Creek.f01 (steady flow) ---

Flow Title=Multiple
Program Version=4.10
Number of Profiles= 7
Profile Names=10-year,25-year,50-year,1pct_min,100-year,1pct_plu,500-year
River Rch & RM=Rocky Cedar Cree,Reach-1         ,122755
     588     783     939     559    1116    2227    1574
River Rch & RM=Rocky Cedar Cree,Reach-1         ,121852
     829    1125    1367     823    1643    3278    2370
River Rch & RM=Rocky Cedar Cree,Reach-1         ,118852
    1040    1426    1745    1057    2110    4210    3083
River Rch & RM=Rocky Cedar Cree,Reach-1         ,117451
    1265    1750    2154    1311    2616    5219    3859
River Rch & RM=Rocky Cedar Cree,Reach-1         ,114359
    1448    2014    2487    1518    3029    6043    4494
River Rch & RM=Rocky Cedar Cree,Reach-1         ,112908
    1609    2244    2775    1696    3383    6751    5031
River Rch & RM=Rocky Cedar Cree,Reach-1         ,111195
    1878    2638    3280    2014    4018    8017    6034
River Rch & RM=Rocky Cedar Cree,Reach-1         ,106407
    2014    2828    3515    2156    4302    8584    6449
River Rch & RM=Rocky Cedar Cree,Reach-1         ,99604
    2650    3759    4703    2902    5790   11552    8781
River Rch & RM=Rocky Cedar Cree,Reach-1         ,91029
    2676    3786    4728    2911    5809   11590    8772
River Rch & RM=Rocky Cedar Cree,Reach-1         ,81832
    2956    4206    5272    3259    6502   12973    9893
River Rch & RM=Rocky Cedar Cree,Reach-1         ,79002
    4096    5883    7422    4612    9202   18361   14152
River Rch & RM=Rocky Cedar Cree,Reach-1         ,68044
    4075    5847    7371    4577    9133   18222   14024
River Rch & RM=Rocky Cedar Cree,Reach-1         ,65202
    4558    6539    8244    5116   10209   20369   15659
River Rch & RM=Rocky Cedar Cree,Reach-1         ,52693
    4644    6661    8394    5208   10391   20732   15925
River Rch & RM=Rocky Cedar Cree,Reach-1         ,46949
    4616    6613    8328    5162   10300   20552   15761
River Rch & RM=Rocky Cedar Cree,Reach-1         ,45768
    4771    6839    8615    5342   10659   21267   16319
River Rch & RM=Rocky Cedar Cree,Reach-1         ,38593
    9160   13267   16839   10504   20959   41819   32450
River Rch & RM=Rocky Cedar Cree,Reach-1         ,37022
    9138   13216   16757   10442   20835   41572   32188
River Rch & RM=Rocky Cedar Cree,Reach-1         ,28087
    9492   13733   17418   10857   21662   43222   33481
River Rch & RM=Rocky Cedar Cree,Reach-1         ,12215
   12820   18647   23744   14853   29635   59129   46108
River Rch & RM=Rocky Cedar Cree,Reach-1         ,6118
   15500   22300   28300   21800   34900   48000   53000
Boundary for River Rch & Prof#=Rocky Cedar Cree,Reach-1         , 1
Up Type= 0
Dn Type= 1
Dn Known WS=390.43
Boundary for River Rch & Prof#=Rocky Cedar Cree,Reach-1         , 2
Up Type= 0
Dn Type= 1
Dn Known WS=391.04
Boundary for River Rch & Prof#=Rocky Cedar Cree,Reach-1         , 3
Up Type= 0
Dn Type= 1
Dn Known WS=391.47
Boundary for River Rch & Prof#=Rocky Cedar Cree,Reach-1         , 4
Up Type= 0
Dn Type= 1
Dn Known WS=391.01
Boundary for River Rch & Prof#=Rocky Cedar Cree,Reach-1         , 5
Up Type= 0
Dn Type= 1
Dn Known WS=391.9
Boundary for River Rch & Prof#=Rocky Cedar Cree,Reach-1         , 6
Up Type= 0
Dn Type= 1
Dn Known WS=392.71
Boundary for River Rch & Prof#=Rocky Cedar Cree,Reach-1         , 7
Up Type= 0
Dn Type= 1
Dn Known WS=393
DSS Import GetInterval= 0
DSS Import GetPeak= 0
DSS Import FillOption= 0

--- Rocky Cedar Creek.g01 (geometry) ---

Geom Title=Existing Conditions
Program Version=4.10

River Reach=Rocky Cedar Cree,Reach-1
Reach XY= 30
        2699726.        6967061.      2707965.67      6957871.17
      2709731.45      6953158.53      2711076.74      6952080.87
      2711022.45      6949912.47      2709375.65      6947631.15
      2710874.24      6944867.13      2708929.45      6942459.52
      2709412.89      6941897.79      2706979.52      6940359.54
      2706422.57      6933862.22      2704719.78      6934953.26
      2700577.37      6929572.52      2702420.54      6929963.47
      2702283.59      6927607.65      2703256.41      6927581.58
       2704174.8      6925650.49       2704133.6      6921657.68
      2706518.27      6918164.65      2705281.83       6913808.7
      2706965.82      6912670.71      2707266.32      6911171.76
      2710728.71      6910005.72      2713470.76      6908305.56
      2714466.15      6906421.47      2715299.52      6906638.31
       2714966.3      6905821.75      2716599.83      6905487.88
      2716478.24      6902466.93      2717701.85      6901183.69

Type RM Length L Ch R = 1 ,122755  ,502,502,502
BEGIN DESCRIPTION:
Rocky Cedar Creek 135.0
END DESCRIPTION:
XS GIS Cut Line= 3
      2700125.99      6967660.96      2699959.29      6966927.57
      2699505.83      6966432.03
#Sta/Elev= 30
  4247.9  557.38  4299.1  555.44  4363.2  555.18  4422.2  552.96  4680.1  550.12
    4718  550.88  4771.4  548.23  4809.3  548.71  4873.4   547.1  4924.7  548.73
  4965.7  546.17    4976  546.98  4991.8  546.49  5005.2  544.77  5005.5  544.27
  5009.2  544.77    5014  546.74  5021.4  546.92  5042.4  546.24  5063.3  547.28
  5070.7  546.28  5240.3  549.65    5297  550.32  5304.4  549.37  5396.3  550.51
  5459.8  553.39  5495.6  552.99  5530.8  554.22  5551.1  553.61  5671.7  556.21
#Mann= 4 ,-1 , 0
  4247.9     .12       0  5005.2     .07       0  5009.2     .12       0
  5551.1     .05       0
Bank Sta=5005.2,5009.2
XS Rating Curve= 0 ,0
Exp/Cntr=0.3,0.1

Type RM Length L Ch R = 1 ,122253  ,401,401,401
BEGIN DESCRIPTION:
Rocky Cedar Creek 134.0
END DESCRIPTION:
XS GIS Cut Line= 3
      2700421.65      6967022.34      2700317.48      6966705.49
      2699776.01      6966411.01
#Sta/Elev= 30
  4797.3  550.09  4840.8  550.96    4904  547.09  4914.5  547.03  4928.9  545.07
  4935.6  545.34  4946.1   543.6  4955.4  545.08  4977.7  544.98  4987.2  545.78
  5009.2   545.8  5040.8  543.67  5056.1   545.2  5082.6  543.99    5104  544.71
  5117.7  539.73  5117.9  539.23  5121.4  539.23  5121.7  539.73    5125  542.77
  5143.9  545.04  5155.8  545.69  5291.7  544.87    5509  547.04    5532  547.82
  5591.9  548.18  5635.6  549.89  5667.5  549.99  5733.4  553.19  5747.2  554.45
#Mann= 4 ,-1 , 0
  4797.3     .12       0  5117.7     .07       0  5121.7     .12       0
    5509     .05       0
Bank Sta=5117.7,5121.7
XS Rating Curve= 0 ,0
Exp/Cntr=0.3,0.1

Type RM Length L Ch R = 1 ,121852  ,272,272,272
BEGIN DESCRIPTION:
Rocky Cedar Creek 133.0
END DESCRIPTION:
XS GIS Cut Line= 3
      2701016.39      6966936.42      2700466.37       6966486.4
      2699826.02      6966311.01
#Sta/Elev= 30
  4301.3  552.31  4319.5  551.23  4426.4  549.84  4455.1  550.38  4482.7  549.06
  4511.1   549.7  4589.4  545.64  4638.9  544.83  4661.2  545.53  4689.4  544.47
  4831.6  545.15  4951.9  543.86  4959.8  544.54  4980.6  542.63    4985  539.24
  4985.3  538.74    4989  539.24  4994.9  540.02  5001.4  543.67    5009  544.03
  5033.1  542.95    5050  544.39  5074.6  543.68  5147.1  546.46  5163.8   545.6
  5292.3  546.37  5385.6  548.48  5416.7  548.26  5503.2  550.97  5675.9  555.86
#Mann= 4 ,-1 , 0
  4301.3     .12       0    4985     .07       0    4989     .12       0
  5503.2     .05       0
Bank Sta=4985,4989
XS Rating Curve= 0 ,0
Exp/Cntr=0.3,0.1

Type RM Length L Ch R = 1 ,121580  ,433,433,433
BEGIN DESCRIPTION:
Rocky Cedar Creek 132.0
END DESCRIPTION:
XS GIS Cut Line= 3
      2701076.01      6966861.01        2700576.        6966261.
        2700276.        6965961.
#Sta/Elev= 30
  4218.7  552.12  4382.1  547.83  4466.7  547.11  4559.1  544.31  4587.8     546
  4637.2  543.13  4786.9   543.8  4807.7  542.56  4815.6  543.21  4822.1  542.25
  4829.9  542.56  4836.4  541.25  4879.3  543.26  4885.8   541.4  4893.7  540.83
    4908  543.19  4943.1  542.54  4963.9   541.1  4978.3  542.98  4990.6  540.07
  4990.8  539.57  4994.6  540.07  4996.5  541.38  5003.3  541.38  5013.9  543.28
    5028  542.49  5056.3  543.75    5099  543.21  5211.9  545.51    5424  551.74
#Mann= 4 ,-1 , 0
  4218.7     .12       0  4990.6     .07       0  4994.6     .12       0
    5099     .05       0
Bank Sta=4990.6,4994.6
XS Rating Curve= 0 ,0
Exp/Cntr=0.3,0.1

Type RM Length L Ch R = 1 ,121147  ,424,424,424
BEGIN DESCRIPTION:
Rocky Cedar Creek 131.0
END DESCRIPTION:
XS GIS Cut Line= 3
      2701326.01      6966561.02        2700826.        6966011.
      2700426.02      6965861.01
#Sta/Elev= 30
  4260.7  550.63  4274.6  550.61  4288.8  549.26  4310.4  548.82  4317.1  549.41
  4381.3  547.44  4423.2  548.11  4451.6  546.65  4494.2  546.46    4530  544.41
  4628.7  543.08  4650.3  544.17  4699.6   542.2  4734.7  543.03  4791.5  540.61
  4819.9  540.85  4848.3  542.57  4890.8  541.13  4982.7   541.6  4990.2  541.49
  5000.6  539.26  5017.2  539.13  5017.4  538.63  5021.2  539.13  5044.1  540.93
  5079.7  542.18  5127.5   542.6  5270.1  547.97  5324.4  547.23  5431.2  550.39
#Mann= 4 ,-1 , 0
  4260.7     .12       0  5017.2     .07       0  5021.2     .12       0
  5127.5     .05       0
Bank Sta=5017.2,5021.2
XS Rating Curve= 0 ,0
Exp/Cntr=0.3,0.1

Type RM Length L Ch R = 1 ,120723  ,380,380,380
BEGIN DESCRIPTION:
Rocky Cedar Creek 130.0
END DESCRIPTION:
XS GIS Cut Line= 3
      2701526.01      6966311.01        2700976.        6965761.
      2700425.97      6965560.99
#Sta/Elev= 30
  4226.7  550.19    4255  548.97  4297.4  549.22  4479.7  545.66  4537.8   546.1
    4552  545.55  4575.2  543.14  4594.4  541.19  4621.5  540.63  4706.2  539.96
  4834.8  540.64    4847   538.9  4847.2   538.4    4851   538.9  4877.3  540.44
  5007.2  539.68  5045.1  540.82  5100.3  540.46  5185.4  541.69  5228.7  543.64
  5253.9  543.37  5340.4  546.55  5345.7  546.12  5355.7  546.98  5419.5  547.75
  5451.4  549.39  5482.7  548.78  5543.9  550.99  5573.8  551.19  5589.8  551.57
#Mann= 8 ,-1 , 0
  4226.7     .05       0  4479.7     .12       0  4575.2     .05       0
  4621.5      .1       0  4706.2     .12       0    4847     .07       0
    4851     .12       0  5573.8     .05       0
Bank Sta=4847,4851
XS Rating Curve= 0 ,0
Exp/Cntr=0.3,0.1

Type RM Length L Ch R = 1 ,120343  ,450,450,450
BEGIN DESCRIPTION:
Rocky Cedar Creek 129.0
END DESCRIPTION:
XS GIS Cut Line= 3
      2701418.46       6965696.7      2701105.96      6965430.98
      2700360.35      6965253.67
#Sta/Elev= 30
  4589.8  547.18  4629.7  544.39  4658.9  540.46  4695.2  540.15  4730.3   538.8
  4735.4  535.61  4735.7  535.11  4739.4  535.61  4744.6  539.02  4779.7  538.49
  4787.5  539.25    4816   538.6  4829.3  539.57  4838.9  539.32    4872  539.03
    4894   539.8  4943.4  538.79  4992.8  540.01  5018.5  539.36  5030.8  537.36
  5051.3  539.13  5133.6  539.74  5226.1  542.43  5308.3  542.72  5462.5  545.88
  5547.1  546.06  5582.1  547.52  5616.7  547.33  5637.2  548.56  5766.4  551.34
#Mann= 6 ,-1 , 0
  4589.8     .05       0  4629.7      .1       0  4735.4     .07       0
  4739.4      .1       0  4838.9     .12       0  5547.1     .05       0
Bank Sta=4735.4,4739.4
XS Rating Curve= 0 ,0
Exp/Cntr=0.3,0.1

Type RM Length L Ch R = 1 ,119893  ,500,500,500
BEGIN DESCRIPTION:
Rocky Cedar Creek 128.0
END DESCRIPTION:
XS GIS Cut Line= 3
      2701651.27      6965417.46      2701394.97      6965079.97
      2700510.77      6965094.52
#Sta/Elev= 30
  4507.5  545.79  4617.2  543.75  4658.4  540.58  4693.8  539.57  4743.7  538.82
  4793.6  539.12  4829.5  537.97  4940.2  537.78  4950.3  537.16  4958.3  532.49
  4958.5  531.99  4962.3  532.49  4970.3  533.59  4980.3  536.87  5030.3  538.02
  5076.8  537.35  5100.3  537.98  5120.3  537.36  5260.3  537.76  5296.5  539.32
  5380.3  539.18  5440.3     541  5550.3  541.83  5580.3  541.25  5593.9  541.93
  5650.3  542.53  5660.3  543.95  5720.4   546.9  5760.4  546.67  5815.6  548.52
#Mann= 6 ,-1 , 0
  4507.5     .05       0  4617.2      .1       0  4958.3     .07       0
  4962.3      .1       0  5076.8     .12       0  5593.9     .05       0
Bank Sta=4958.3,4962.3
XS Rating Curve= 0 ,0
Exp/Cntr=0.3,0.1

Type RM Length L Ch R = 1 ,119393  ,541,541,541
BEGIN DESCRIPTION:
Rocky Cedar Creek 127.0
END DESCRIPTION:
XS GIS Cut Line= 3
      2702101.03      6965386.03       2701419.7      6964612.78
       2700249.9       6964871.2
#Sta/Elev= 30
  3969.4  542.62  4161.1  540.93  4210.4  541.67  4302.4  540.12  4373.6  540.99
  4465.6   539.4  4529.2  540.41  4586.1  537.83    4638  538.32  4805.2  535.51
  4833.7   537.3  4890.6  534.94  4911.5  536.72  4968.4   536.2  4975.7  535.89
  4980.3  532.56  4980.8  532.06  4984.9  532.56    4999  536.61  5011.9  537.19
  5085.7  536.41  5172.4  537.64  5196.8  538.67  5250.7  536.76    5352  538.29
  5372.5  539.61  5403.2   538.4  5536.3  538.81  5778.6  542.89    6198  552.33
#Mann= 6 ,-1 , 0
  3969.4     .05       0    4638      .1       0  4980.3     .07       0
  4984.9      .1       0  5172.4     .12       0  5778.6     .05       0
Bank Sta=4980.3,4984.9
XS Rating Curve= 0 ,0
Exp/Cntr=0.3,0.1

Type RM Length L Ch R = 1 ,118852  ,484,484,484
BEGIN DESCRIPTION:
Rocky Cedar Creek 126.0
END DESCRIPTION:
XS GIS Cut Line= 3
      2702151.01      6965186.03      2701805.62      6964330.84
      2700700.99        6964036.
#Sta/Elev= 30
  4077.7  540.67  4185.1  541.32  4255.7  539.62  4340.7  541.53  4453.4  538.13
  4507.1  541.14  4531.2  538.23  4731.6  535.46  4751.8  536.57  4775.4  534.64
  4838.2  535.62  5007.6  533.92  5008.1  533.42  5012.3  533.92  5030.7  535.46
  5113.5  534.82  5200.8  536.58  5217.4  537.15  5227.3  535.37  5252.3  536.83
  5294.6  535.13  5475.7   536.8  5765.5  542.69    5798  544.72  5832.9   544.8
  5879.4     548  5941.5  547.27  6013.9  551.59  6034.6  554.56  6143.3   556.9
#Mann= 7 ,-1 , 0
  4077.7      .1       0  4731.6     .12       0  4838.2      .1       0
  5007.6     .07       0  5012.3      .1       0  5200.8     .12       0
  5294.6     .05       0
Bank Sta=5007.6,5012.3
XS Rating Curve= 0 ,0
Exp/Cntr=0.3,0.1

Type RM Length L Ch R = 1 ,118368  ,359,359,359
BEGIN DESCRIPTION:
Rocky Cedar Creek 125.0
END DESCRIPTION:
XS GIS Cut Line= 3
      2702551.21      6965421.27      2701985.98      6963950.98
      2701175.97      6963760.99
#Sta/Elev= 30
  3424.8  542.57  3500.1  540.77  3761.9  539.81  3864.3  538.63  3917.9  540.26
  3979.8  537.53  4015.2  538.93  4069.8  537.73  4124.5  540.46  4142.9  537.86
  4159.2  537.42  4179.1  537.15  4203.1  539.69  4228.4     540  4271.5   537.8
  4356.5  538.35  4452.4   536.3  4487.7  537.03  4542.4  534.39  4636.7  532.94
    4644  532.52  4644.5  532.02  4648.7  532.52  4766.4  534.71  4796.4  533.38
  5127.8  533.84  5265.3  534.48  5633.3  538.69  5770.9  544.11    5832  558.62
#Mann= 10 ,-1 , 0
  3424.8     .05       0  3761.9      .1       0  4159.2     .12       0
  4203.1      .1       0  4356.5     .12       0  4636.7      .1       0
    4644     .07       0  4648.7      .1       0  5127.8     .12       0
  5265.3     .05       0
Bank Sta=4644,4648.7
XS Rating Curve= 0 ,0
Exp/Cntr=0.3,0.1

Type RM Length L Ch R = 1 ,118009  ,558,558,558
BEGIN DESCRIPTION:
Rocky Cedar Creek 124.0
END DESCRIPTION:
XS GIS Cut Line= 3
      2703356.77      6964789.32        2702276.        6963761.
      2701300.97      6963285.98
#Sta/Elev= 30
  3508.4  545.28  3613.9  542.04  3719.9   540.6  3783.7  541.28  3889.7  538.72
  3939.1  539.33    4003  537.14  4076.9  538.16  4117.4  538.64  4165.6  537.98
  4222.2  534.96  4379.6  534.63  4420.4  533.34  4490.8  533.68  4547.4  531.38
  4653.8  532.65  4735.9  530.63  4736.5  530.13  4740.7  530.63  4802.2  532.36
    5003  532.74  5022.5   531.6  5089.2   533.3  5393.4  533.97  5628.4  535.38
  5808.7  541.32    5927  542.42  6011.6  547.44  6045.8  546.75  6084.8  548.22
#Mann= 7 ,-1 , 0
  3508.4     .05       0  4076.9     .12       0  4117.4     .05       0
  4379.6      .1       0  4735.9     .07       0  4740.7      .1       0
  5393.4     .05       0
Bank Sta=4735.9,4740.7
XS Rating Curve= 0 ,0
Exp/Cntr=0.3,0.1

Type RM Length L Ch R = 1 ,117451  ,324,324,324
BEGIN DESCRIPTION:
Rocky Cedar Creek 123.0
END DESCRIPTION:
XS GIS Cut Line= 3
      2703826.03      6964661.03      2702675.58      6963390.76
      2701825.96      6962710.97
#Sta/Elev= 30
  3286.2   549.5  3406.9  546.88  3527.2  545.94  3597.5  543.41  3725.2  543.48
  3859.7  540.16    3909  541.13  3959.1  539.63  4121.9  538.22  4149.7  538.98
  4211.8  537.54  4438.6  535.99    4518  534.94  4581.5   536.1  4624.1  533.92
  4678.1  533.16  4801.2   530.6  4819.8  529.19  4820.8  528.69  4825.8  529.19
  4829.5  530.14  4921.5  531.27  4985.7  529.67  5091.6   531.5  5197.1  531.53
  5469.1  533.46  5717.5  535.42  5767.9  538.72  5867.9  541.39  6088.1   549.9
#Mann= 8 ,-1 , 0
  3286.2     .05       0  4211.8     .12       0  4438.6     .05       0
  4678.1      .1       0  4819.8     .07       0  4825.8      .1       0
  5197.1     .12       0  5469.1     .05       0
Bank Sta=4819.8,4825.8
XS Rating Curve= 0 ,0
Exp/Cntr=0.3,0.1

Type RM Length L Ch R = 1 ,117127  ,453,453,453
BEGIN DESCRIPTION:
Rocky Cedar Creek 122.0
END DESCRIPTION:
XS GIS Cut Line= 3
      2703726.01      6964361.01        2702926.        6963261.
      2702176.01      6962511.01
#Sta/Elev= 30
  3634.6  545.47  3706.9  543.17  3949.5  540.83  4029.1  538.64  4265.2  537.99
  4292.7  536.57  4415.2  536.41    4659  534.53  4660.4  534.34  4700.7  532.64
  4730.1   533.2  4772.2  530.68  4916.3  530.58  4945.3  529.31  4987.4  529.34
  4988.7  528.09  4989.7  527.59  4994.7  528.09  5051.3  530.44  5138.5  530.23
  5175.7  530.44  5261.3  530.89  5317.4  530.71    5428  531.35  5467.2  531.57
  5772.6  535.79  5829.1   538.1    5914  543.66  5970.6  545.61  6055.4  546.76
#Mann= 12 ,-1 , 0
  3634.6     .05       0  4415.2     .12       0    4659     .05       0
  4660.4      .1       0  4988.7     .07       0  4994.7      .1       0
  5138.5     .12       0  5175.7     .05       0  5261.3     .12       0
  5317.4     .05       0    5428     .12       0  5467.2     .05       0
Bank Sta=4988.7,4994.7
XS Rating Curve= 0 ,0
Exp/Cntr=0.3,0.1

Type RM Length L Ch R = 1 ,116674  ,563,563,563
BEGIN DESCRIPTION:
Rocky Cedar Creek 121.0
END DESCRIPTION:
XS GIS Cut Line= 3
      2703926.01      6963961.02        2703226.        6962961.
      2702226.01        6962461.
#Sta/Elev= 30
  3784.9  542.79  3870.4  541.23  3943.6   541.4  4057.4  537.05  4122.8  537.45
  4173.4  535.79    4346  534.54  4444.5  532.38  4581.4  533.67  4670.4  531.45
  4779.2  528.56  4946.4  529.99  4992.1  529.75  4998.2  529.02  4999.5  527.61
  5000.5  527.11  5005.6  527.61  5019.6  529.14    5081  530.38  5176.1  529.38
  5327.5  530.05  5519.9  530.43  5846.9  537.06    5914  537.45  5953.1  540.45
  5958.7  539.93  5975.5  542.42  6070.5   544.6  6087.3  546.34  6123.6  546.25
#Mann= 7 ,-1 , 0
  3784.9     .05       0  4670.4     .12       0  4779.2      .1       0
  4946.4     .12       0  4999.5     .07       0  5005.6     .12       0
  5327.5     .05       0
Bank Sta=4999.5,5005.6
XS Rating Curve= 0 ,0
Exp/Cntr=0.3,0.1

Type RM Length L Ch R = 1 ,116111  ,486,486,486
BEGIN DESCRIPTION:
Rocky Cedar Creek 120.0
END DESCRIPTION:
XS GIS Cut Line= 3
      2703950.99      6963585.96      2703706.27      6962731.51
      2702326.04      6962361.01
#Sta/Elev= 30
  4111.2   539.8  4230.8  538.68    4262  539.63    4314  537.62  4469.6  535.94
    4522  533.78  4626.1   532.6  4646.9  533.48  4731.9  531.56  4823.7   532.1
  4910.1  529.77  4958.9  527.12  4969.3  527.77  4980.8  524.47  4981.8  523.97
    4987  524.47  4990.1   527.8  5063.7  529.54  5279.8  527.93  5331.5  528.93
  5370.7  528.44  5682.1  529.46  5686.3  529.52  5766.5  528.77  5947.3  531.92
    6097  537.37  6201.3  538.69  6336.9   542.1  6398.1  544.91  6429.1  544.45
#Mann= 8 ,-1 , 0
  4111.2     .05       0  4910.1      .1       0  4980.8     .07       0
    4987      .1       0  5331.5     .12       0  5370.7      .1       0
  5682.1     .12       0  5686.3     .05       0
Bank Sta=4980.8,4987
XS Rating Curve= 0 ,0
Exp/Cntr=0.3,0.1

Type RM Length L Ch R = 1 ,115625  ,359,359,359
BEGIN DESCRIPTION:
Rocky Cedar Creek 119.0
END DESCRIPTION:
XS GIS Cut Line= 4
      2704782.96      6963481.99      2703915.68      6962302.16
       2703806.3      6962305.64      2702361.15      6962041.06
#Sta/Elev= 30
  3496.4  543.98  3545.7  545.36  3696.2  539.11  3857.6  535.02  4159.9  530.21
  4195.4  531.26  4239.3  529.98  4339.6  530.87  4630.7  528.98    4797  528.39
  4990.4  528.37  5000.4  525.85  5007.3   521.8  5008.3   521.3  5013.5   521.8
  5030.4  526.76  5080.6   528.5  5192.4   527.2  5324.6  528.49  5334.8  527.32
  5342.8  528.48  5455.4  529.02  5765.2  530.31  5839.3  529.98  6239.6  534.12
  6345.8  536.28  6381.9  538.43  6457.2  538.48  6510.4  541.78  6539.3  540.85
#Mann= 9 ,-1 , 0
  3496.4     .12       0  3857.6      .1       0  4630.7     .12       0
    4797      .1       0  5007.3     .07       0  5013.5      .1       0
  5455.4     .12       0  5765.2      .1       0  5839.3     .05       0
Bank Sta=5007.3,5013.5
XS Rating Curve= 0 ,0
Exp/Cntr=0.3,0.1

Type RM Length L Ch R = 1 ,115266  ,442,442,442
BEGIN DESCRIPTION:
Rocky Cedar Creek 118.0
END DESCRIPTION:
XS GIS Cut Line= 3
      2704976.03      6962811.02        2703976.        6962011.
      2703322.82      6961659.32
#Sta/Elev= 30
    3715   541.5  3800.7  538.55  3920.7  537.42  3978.4  534.12  4035.2  533.35
    4092  535.05  4170.5  531.94  4314.2  529.74  4405.8  530.27    4433  528.06
  4540.2  525.52    4593  527.38  4602.5   527.4  4697.1   528.6  4753.1   526.9
  4953.2  527.75  5009.5  526.08  5022.5  522.83  5023.5  522.33  5028.8  522.83
  5031.4  525.68  5053.3  527.77  5113.3  526.39  5356.5  528.12  5467.5  528.49
  5586.2  530.51  5643.9  532.79  5676.3  535.78  5735.6  537.08  5737.5  537.08
#Mann= 9 ,-1 , 0
    3715     .12       0  4314.2      .1       0    4593     .12       0
  4602.5      .1       0  5022.5     .07       0  5028.8      .1       0
  5356.5     .12       0  5467.5     .05       0  5735.6     .12       0
Bank Sta=5022.5,5028.8
XS Rating Curve= 0 ,0
Exp/Cntr=0.3,0.1

Type RM Length L Ch R = 1 ,114824  ,465,465,465
BEGIN DESCRIPTION:
Rocky Cedar Creek 117.0
END DESCRIPTION:
XS GIS Cut Line= 3
      2705325.99      6962710.99        2704126.        6961611.
      2703575.99      6961060.99
#Sta/Elev= 30
  3376.8  542.07  3511.5   541.2  3688.5  536.45  3893.2  535.87  3957.3  533.35
  3992.5   535.1  4134.3  532.06  4289.7  532.82  4431.5  527.24  4490.9  528.74
  4551.8  525.34    4672  525.99  4686.2  522.97    4693  526.52  4749.7  523.58
  4792.2  526.23    4841     526  4874.1  526.02  4989.7  525.68  5018.8  527.34
  5029.2  524.87  5043.4  521.72  5044.5  521.22  5050.7  521.72  5061.2  525.42
  5103.7  526.88  5256.7  526.67  5400.7  527.32  5463.9  530.72  5782.5  548.05
#Mann= 10 ,-1 , 0
  3376.8     .12       0  4490.9      .1       0    4841     .12       0
  4874.1      .1       0  4989.7     .12       0  5029.2      .1       0
  5043.4     .07       0  5050.7      .1       0  5256.7     .12       0
  5463.9     .05       0
Bank Sta=5043.4,5050.7
XS Rating Curve= 0 ,0
Exp/Cntr=0.3,0.1

Type RM Length L Ch R = 1 ,114359  ,549,549,549
BEGIN DESCRIPTION:
Rocky Cedar Creek 116.0
END DESCRIPTION:
XS GIS Cut Line= 3
      2705376.02      6962461.02        2704376.        6961261.
      2703481.09      6960855.93
#Sta/Elev= 30
  3428.5   538.9    3493  539.94  3548.9  537.03  3754.6  536.82  3805.4  534.36
  3996.7  532.92  4046.2  534.81  4074.8  532.39  4294.8  530.01  4379.4  531.37
    4564  526.34  4654.9  524.45  4685.3  522.33  4759.9  523.92  4784.3  522.61
  4983.4   525.2  4993.3   523.8  4995.7  521.56  4996.8  521.06  5003.1  521.56
  5022.5  525.34  5069.1  524.81  5311.3  525.32  5586.8  533.09  5671.1  537.93
  5707.8  537.52    5748  539.77  5800.2  546.79  5868.7  548.35  5972.9  546.99
#Mann= 8 ,-1 , 0
  3428.5     .12       0    4564      .1       0  4654.9     .12       0
  4759.9      .1       0  4995.7     .07       0  5003.1      .1       0
  5069.1     .12       0  5311.3     .05       0
Bank Sta=4995.7,5003.1
XS Rating Curve= 0 ,0
Exp/Cntr=0.3,0.1

Type RM Length L Ch R = 1 ,113810  ,312,312,312
BEGIN DESCRIPTION:
Rocky Cedar Creek 115.0
END DESCRIPTION:
XS GIS Cut Line= 3
      2705286.96      6962185.22      2704613.36      6960855.38
      2703814.78      6960393.59
#Sta/Elev= 30
    3523  535.91  3584.9  536.47  3629.5  533.94    3713  533.21  3796.5  535.13
  3846.6  532.04  3964.9   530.4  4032.2  532.16    4077  530.16  4113.9  532.07
  4314.4  527.87  4353.3  528.84  4375.9  527.42  4559.4  525.47  4598.4  523.61
  4599.5  521.55  4600.8  521.05  4608.4  521.55  4687.5  523.69    4716  521.62
    4732  521.56  4748.7  523.48  4939.1  522.71  5254.8  524.27  5484.3  526.72
  5608.7  530.65  5673.3  534.53  5769.4  534.46  5849.8  540.97  5936.2  541.64
#Mann= 6 ,-1 , 0
    3523     .12       0  4375.9      .1       0  4599.5     .05       0
  4608.4      .1       0  4939.1     .12       0  5254.8     .05       0
Bank Sta=4599.5,4608.4
XS Rating Curve= 0 ,0
Exp/Cntr=0.3,0.1

Type RM Length L Ch R = 1 ,113498  ,590,590,590
BEGIN DESCRIPTION:
Rocky Cedar Creek 114.0
END DESCRIPTION:
XS GIS Cut Line= 3
       2706029.8      6962659.42        2704876.        6960711.
      2704275.97      6960160.97
#Sta/Elev= 30
  2735.6  541.21  2741.2  541.08  2810.5  543.21  3007.4   539.3  3081.6  541.06
  3167.3  538.05  3210.3  540.21  3395.5   535.5  3453.9  538.18  3767.8   531.3
  4023.3  530.66  4211.9  527.03  4268.8   527.1  4300.1  524.16    4380  527.96
  4475.6  523.44  4616.2   524.2  4716.7  521.31    4718  520.81  4725.6  521.31
  4758.2  523.56  4789.5  521.57  4810.9  523.43  4934.3  522.03  5269.2  522.46
    5432  526.36  5509.7  529.55    5559  535.61  5615.7  539.47    5814  548.23
#Mann= 7 ,-1 , 0
  2735.6      .1       0  2741.2     .12       0  4211.9     .03       0
  4616.2     .03       0  4716.7     .03       0  4725.6     .03       0
  4934.3     .05       0
Bank Sta=4716.7,4725.6
XS Rating Curve= 0 ,0
Exp/Cntr=0.3,0.1

Type RM Length L Ch R = 1 ,112908  ,605,605,605
BEGIN DESCRIPTION:
Mapping XS 0f116183
END DESCRIPTION:
XS GIS Cut Line= 3
      2706692.76      6961890.04      2705346.87      6960388.36
      2704522.35      6959845.92
#Sta/Elev= 30
  2984.4   543.7  3158.7  540.78    3194  542.78  3271.8  538.52  3342.8   540.5
  3363.7  537.38  3392.1  536.35  3463.2  536.73  3561.8  534.36  3611.9  535.89
  3682.2  532.51  3718.1  533.41  3788.8  531.47    3831  533.25  3965.5  528.32
  4015.6  530.49  4071.7  526.05  4121.1  525.74  4327.8  524.74    4589  521.51
  4609.9  522.64  4869.4  521.59  4964.3   522.7  5326.9  521.29  5328.3  520.79
    5337  521.29  5432.2  522.47    5433  522.49  5744.1   529.5  5987.9  541.71
#Mann= 9 ,-1 , 0
  2984.4      .1       0  3158.7     .12       0  4121.1      .1       0
  4327.8     .12       0  4869.4     .03       0  5326.9     .03       0
    5337     .03       0  5432.2     .12       0    5433     .05       0
Bank Sta=5326.9,5337
XS Rating Curve= 0 ,0
Exp/Cntr=0.3,0.1

Type RM Length L Ch R = 1 ,112303  ,547,547,547
BEGIN DESCRIPTION:
Mapping XS e014ce85
END DESCRIPTION:
XS GIS Cut Line= 3
      2706844.26      6961291.13      2705819.96      6960045.48
      2705207.95      6959411.77
#Sta/Elev= 30
  3402.8  538.77  3466.1  538.55  3522.1  536.91  3529.9  537.71  3608.1  534.44
  3664.1  536.25  3700.7  532.86  3707.1  533.82  3750.2  532.59  3756.7  534.15
  3801.8  532.61  3856.1   532.7  3898.7  530.29  3976.9  529.07  4040.8  526.63
  4055.1  527.04  4104.6  524.86  4380.5  522.68  4420.3  521.38  4421.7  520.88
  4430.4  521.38  4431.8  522.37  4436.4  522.27  4460.5  523.02  4503.4  521.63
  5537.7  522.38  5587.3  526.26  5707.4   530.5  5728.8   532.8  5896.5  540.99
#Mann= 6 ,-1 , 0
  3402.8     .05       0  3801.8      .1       0  4380.5     .03       0
  4420.3     .03       0  4430.4     .03       0  4436.4     .05       0
Bank Sta=4420.3,4430.4
XS Rating Curve= 0 ,0
Exp/Cntr=0.3,0.1

Type RM Length L Ch R = 1 ,111756  ,467,467,467
BEGIN DESCRIPTION:
Mapping XS d9230bea
END DESCRIPTION:
XS GIS Cut Line= 3
      2707197.59      6961052.46      2706249.65      6959729.51
      2705201.03      6959036.02
#Sta/Elev= 30
  3377.8   542.7  3387.4  541.33  3502.6  538.11  3701.9  535.47  3731.3  534.19
  3752.2  534.71    3767  533.76  3773.3  532.03  3787.9   532.3  3796.4  534.34
  3810.2   534.3  3924.2  530.53  3953.7   530.1  3959.8  531.25  4117.7  527.46
  4167.4   527.5  4196.9  526.34  4217.8  523.82  4282.8  521.62  4303.7  522.65
  4354.1  521.62  5615.9  521.57  5617.3  521.07  5626.4  521.57  5648.6  525.49
  5693.1  526.76  5720.9  529.19  5735.9  528.64    5778  531.75  6262.5  544.18
#Mann= 3 ,-1 , 0
  3377.8     .03       0  5615.9     .03       0  5626.4     .03       0
Bank Sta=5615.9,5626.4
XS Rating Curve= 0 ,0
Exp/Cntr=0.3,0.1

Type RM Length L Ch R = 1 ,111289  ,94,94,94
BEGIN DESCRIPTION:
Mapping XS 9729893c
END DESCRIPTION:
XS GIS Cut Line= 4
      2707552.56      6960381.49      2706615.05      6959464.82
      2706161.93      6959006.48      2705551.03      6958586.02
#Sta/Elev= 30
  3695.3  538.17  3940.8  533.56  4060.9   529.5  4117.5   529.2    4259  525.09
  4411.2  523.52  4503.7  522.93  4516.3  522.68  4639.1  521.78  5052.7  521.29
  5054.1  520.79  5063.3  521.29    5157  522.29  5241.9  521.41    5355  523.06
  5376.2  522.12  5475.2  522.86  5510.6  522.06  5723.7  529.31  5831.2  535.21
  5846.1  534.33    5861  530.28  5911.7   529.8  6046.7  531.12  6061.2  531.84
  6083.1  536.48  6177.6  535.08  6270.2  537.02  6285.1  535.99  6392.6  537.82
#Mann= 7 ,-1 , 0
  3695.3     .05       0  4411.2     .12       0  4503.7     .05       0
  4516.3     .03       0  4639.1     .03       0  5052.7     .03       0
  5063.3     .03       0
Bank Sta=5052.7,5063.3
XS Rating Curve= 0 ,0
Exp/Cntr=0.3,0.1

Type RM Length L Ch R = 1 ,111195  ,137,137,137
BEGIN DESCRIPTION:
Mapping XS 5e7a3c91
END DESCRIPTION:
XS GIS Cut Line= 6
       2707661.9      6960371.04      2707417.14      6960136.69
      2707047.35      6959772.11       2706391.1      6959126.27
      2706104.64      6958865.86      2705730.36      6958631.93
#Sta/Elev= 30
  3659.6  538.59  3854.8  535.95    3890  537.84  3897.2  535.61  3904.1  537.96
  3939.7  536.18  3946.6   538.1  4034.7   538.2  4072.8  537.98  4616.1  538.03
  4749.2  538.25  5580.5  538.11  5608.4  538.02  5615.8  535.74  5622.6  537.75
  5700.9  535.87  5721.9  537.76  5736.1  533.03  5742.8  535.47  5750.3  533.14
    5757  536.12  5778.7  534.26  5825.5  537.94  5900.8  537.01  5906.7  533.12
    5922  531.27  5975.9  530.36  6104.8  531.53  6131.9  536.76    6267  536.01
#Mann= 7 ,-1 , 0
  3659.6     .05       0  4034.7      .1       0  4072.8     .05       0
  4616.1     .12       0  4749.2     .05       0  5900.8     .04       0
  6131.9     .05       0
Bank Sta=5900.8,6131.9
XS Rating Curve= 0 ,0
Exp/Cntr=0.3,0.1

Type RM Length L Ch R = 1 ,111058  ,858,858,858
BEGIN DESCRIPTION:
Mapping XS 9d3a723d
END DESCRIPTION:
XS GIS Cut Line= 3
      2707717.49      6960330.71      2706806.03      6959341.12
      2705869.75       6958592.1
#Sta/Elev= 30
  3647.2   538.9  3669.3  538.49  3736.5  537.16  3805.4  536.15    3879  534.13
  3941.4  533.19  4163.9  528.29  4213.5   528.3  4306.4  527.03  4349.6  526.72
  4448.9  523.66  4519.1   524.6  4773.5  522.32  4857.1  517.33  4893.7  516.15
  4914.7  515.95  4943.1   519.8  4973.4  509.79  4974.9  509.29  4984.1  509.79
  5015.4  516.03  5518.5  519.51    5669  525.73  5675.4  528.26  5710.6  530.16
  5875.5  533.94  6088.4   531.7  6102.8  532.29  6138.1  540.97  6191.6  539.05
#Mann= 17 ,-1 , 0
  3647.2     .05       0  3669.3     .12       0  3736.5     .05       0
  3805.4     .12       0    3879     .05       0  3941.4      .1       0
  4163.9     .05       0  4213.5     .12       0  4306.4     .05       0
  4349.6      .1       0  4448.9     .05       0  4519.1     .12       0
  4857.1     .05       0  4893.7      .1       0  4973.4     .07       0
  4984.1      .1       0  5015.4     .05       0
Bank Sta=4973.4,4984.1
XS Rating Curve= 0 ,0
Exp/Cntr=0.3,0.1

Type RM Length L Ch R = 1 ,110200  ,523,523,523
BEGIN DESCRIPTION:
Mapping XS 8836f8a1
END DESCRIPTION:
XS GIS Cut Line= 3
      2708124.64      6959859.71      2707129.85      6958693.05
       2706140.6      6958380.65
#Sta/Elev= 30
  3437.4  538.94  3488.6  537.51  3608.1  535.21  3747.9  531.63  4034.2  524.71
  4144.7  521.88    4365  518.24  4717.6  516.82  4975.2  515.76  4997.4  511.92
  5011.1  505.46  5012.6  504.96  5022.1  505.46  5024.5     507  5037.6  507.79
  5056.9  514.12    5069  516.26    5259  515.21  5330.3  516.82  5390.7   516.2
  5461.4  517.74  5562.8  520.07  5589.9  522.45  5627.5  523.09  5635.3  524.62
  5645.8  523.57  5666.8  525.47  5742.1  527.13  5961.3  533.24    6008  536.44
#Mann= 13 ,-1 , 0
  3437.4     .12       0  3488.6      .1       0  3608.1     .12       0
  3747.9      .1       0  4034.2     .12       0  4144.7      .1       0
  4717.6     .12       0  5011.1     .07       0  5022.1     .12       0
    5259      .1       0  5330.3     .12       0  5461.4      .1       0
  5742.1     .05       0
Bank Sta=5011.1,5022.1
XS Rating Curve= 0 ,0
Exp/Cntr=0.3,0.1

Type RM Length L Ch R = 1 ,109677  ,613,613,613
BEGIN DESCRIPTION:
Mapping XS 9cdc526f
END DESCRIPTION:
XS GIS Cut Line= 3
      2708572.57      6959297.22      2707499.65      6958469.09
       2706775.7      6958172.22
#Sta/Elev= 30
  3616.3  538.93  3896.4  533.71  3910.9  533.18  3917.2  530.03  3946.2  529.35
  3960.7  534.46  3981.5  534.58  4016.8   528.8  4396.9  520.44  4477.6  519.49
  4507.7  518.65  4723.3  515.95  4838.3  514.35  4846.1  514.28    4880  513.79
  4887.8  510.65  4894.5  513.67    4938   515.5  4958.8  505.78  4965.1  508.17
  4974.9  504.82  4976.4  504.32  4985.9  504.82  4986.4  510.07  5001.5  513.97
  5031.5  515.38  5217.5  513.81    5555  525.35  5711.2  534.83  5754.1   537.4
#Mann= 14 ,-1 , 0
  3616.3     .05       0  4396.9     .12       0  4477.6      .1       0
  4507.7     .12       0  4723.3      .1       0  4838.3     .12       0
  4846.1      .1       0  4974.9     .07       0  4985.9      .1       0
  5001.5     .12       0  5031.5      .1       0  5217.5     .12       0
    5555      .1       0  5711.2     .12       0
Bank Sta=4974.9,4985.9
XS Rating Curve= 0 ,0
Exp/Cntr=0.3,0.1

Type RM Length L Ch R = 1 ,109064  ,665,665,665
BEGIN DESCRIPTION:
Mapping XS 2894b873
END DESCRIPTION:
XS GIS Cut Line= 3
      2708215.75      6958509.86      2707569.09      6958049.82
       2706940.4      6958002.13
#Sta/Elev= 30
  4212.2  525.46  4224.6  522.17  4239.3  520.46    4267  520.33    4275     521
  4319.3  518.27  4527.8  516.05  4641.4  514.45    4655  513.45  4669.7  509.06
  4684.5  514.21  4690.6  514.49  4741.1  513.18  4850.1  514.38  4862.8   514.1
  4877.6  511.46    4911  514.44  4985.1  514.67  4993.2     513  4999.1   504.7
  5000.6   504.2  5010.1   504.7  5018.9   506.9    5029  514.71  5079.1  514.05
  5191.5  516.62  5229.5  519.61  5269.7  520.21  5414.7   530.6  5636.3  538.66
#Mann= 7 ,-1 , 0
  4212.2     .05       0    4267     .12       0  4527.8      .1       0
    4911     .12       0  4999.1     .07       0  5010.1     .12       0
  5414.7      .1       0
Bank Sta=4999.1,5010.1
XS Rating Curve= 0 ,0
Exp/Cntr=0.3,0.1

Type RM Length L Ch R = 1 ,108399  ,146,146,146
BEGIN DESCRIPTION:
Mapping XS 4c7bd7d5
END DESCRIPTION:
XS GIS Cut Line= 3
      2708911.08      6958344.08      2707994.44      6957693.05
      2706979.95      6957823.11
#Sta/Elev= 30
  3875.4  535.86  3918.6   534.1  4096.4  529.62    4176  529.54  4390.4  523.01
  4433.6  523.65  4440.8  522.24  4561.8  520.87  4853.5  515.12  4948.8  513.21
  4972.2  514.08  4978.4  513.47  4985.5  508.06  4987.6  503.94  4989.1  503.44
  4998.7  503.94  5008.2  507.96  5018.1  509.79  5023.1  508.55  5029.2  511.21
  5035.4  512.25  5088.9   513.6  5243.4  513.43    5393  512.84    5505  515.67
  5538.1  516.99  5613.1  519.21    5753  526.38  5818.8  528.71  6022.5  534.53
#Mann= 14 ,-1 , 0
  3875.4      .1       0  3918.6     .12       0  4561.8     .05       0
  4853.5     .12       0  4987.6     .07       0  4998.7     .12       0
  5029.2      .1       0  5035.4     .12       0  5243.4      .1       0
    5393     .12       0    5505      .1       0  5538.1     .12       0
    5753      .1       0  5818.8     .12       0
Bank Sta=4987.6,4998.7
XS Rating Curve= 0 ,0
Exp/Cntr=0.3,0.1

Type RM Length L Ch R = 1 ,108253  ,563,563,563
BEGIN DESCRIPTION:
Mapping XS 4ce398d8
END DESCRIPTION:
XS GIS Cut Line= 3
      2708667.17      6957945.65       2708011.8      6957546.35
      2707035.27      6957555.03
#Sta/Elev= 30
  4255.8  526.54  4348.1  525.35  4412.1  522.22  4528.3  521.41  4586.4  518.87
  4617.3  518.45  4644.5  519.83  4754.8  515.86  4824.5  514.69  4892.4  514.22
  4929.1  512.14  4965.9  513.79  5002.7  509.34  5008.6  507.31  5012.2  503.99
  5013.8  503.49  5023.4  503.99  5029.3  504.21    5039  510.94    5049  512.66
    5088  513.07  5258.3  512.42  5511.2   514.3  5609.1  515.88  5639.1  517.76
  5719.1  518.52  5839.1  523.66  5879.1  522.88  5919.1  524.91  5999.8  526.45
#Mann= 8 ,-1 , 0
  4255.8     .05       0  4824.5     .12       0  5012.2     .07       0
  5023.4     .12       0  5029.3      .1       0    5088     .12       0
  5258.3      .1       0  5511.2     .12       0
Bank Sta=5012.2,5023.4
XS Rating Curve= 0 ,0
Exp/Cntr=0.3,0.1

Type RM Length L Ch R = 1 ,107690  ,859,859,859
BEGIN DESCRIPTION:
Mapping XS 1e9ee2f2
END DESCRIPTION:
XS GIS Cut Line= 4
      2708714.94      6957759.04       2708098.6      6957281.59
      2707727.88      6957205.06      2707159.69      6956829.26
#Sta/Elev= 30
  4225.6  528.17    4826  513.29  4850.2  512.78  4942.5  512.23  4979.3  513.67
  4985.6  509.97  4988.2  504.69  4989.7  504.19  4999.4  504.69  5069.2  513.05
  5180.3  511.19  5222.3  508.36  5229.1  511.79  5280.9  511.76    5304  511.28
  5324.4  506.02  5329.6   506.2  5334.7   512.1  5381.5  512.24  5396.1  508.33
  5424.5  512.56    5446  509.67  5468.3  513.31  5474.3  511.03  5504.4  511.23
  5567.6  518.67  5589.8  517.27  5625.8  520.93  5814.4  521.49    6065  530.25
#Mann= 10 ,-1 , 0
  4225.6     .05       0    4826     .12       0  4850.2      .1       0
  4942.5     .12       0  4988.2     .07       0  4999.4     .12       0
  5180.3      .1       0  5280.9     .12       0  5381.5      .1       0
  5424.5     .05       0
Bank Sta=4988.2,4999.4
XS Rating Curve= 0 ,0
Exp/Cntr=0.3,0.1

Type RM Length L Ch R = 1 ,106831  ,424,424,424
BEGIN DESCRIPTION:
Mapping XS 91ed82e5
END DESCRIPTION:
XS GIS Cut Line= 3
      2708706.22       6957372.7      2708315.62      6956717.35
      2708060.27      6956427.38
#Sta/Elev= 30
  4241.4   525.5    4418  520.18  4462.6     518    4702  513.14  4744.8  511.72
  4760.4  511.88  4781.8  510.96  4797.4  511.22  4851.3  510.04  4861.6  510.97
  4914.2   509.2  4951.2  509.85  4957.9  509.32  4978.4   503.6  4982.5  503.08
    4984  502.58    4994  503.08  4999.3   507.3  5008.7  507.36  5065.6  511.14
  5079.4   511.1  5129.2  516.05  5192.8  518.85  5227.9  521.59  5235.5  521.38
  5270.6  523.39  5348.4  525.55  5355.9  526.65  5384.4  528.01  5390.7  527.68
#Mann= 5 ,-1 , 0
  4241.4     .05       0  4851.3     .12       0  4957.9     .05       0
  4982.5     .04       0    4994     .05       0
Bank Sta=4982.5,4994
XS Rating Curve= 0 ,0
Exp/Cntr=0.3,0.1

Type RM Length L Ch R = 1 ,106407  ,660,660,660
BEGIN DESCRIPTION:
Mapping XS ba9696f6
END DESCRIPTION:
XS GIS Cut Line= 3
      2708931.28       6956811.1      2708676.08      6956545.48
      2708181.28      6956292.87
#Sta/Elev= 30
  4631.4  521.78  4705.9  519.41  4868.5  511.63  4908.6  510.79  4946.5  510.85
  4974.8  509.74    4990  501.13  4991.6  500.63  5001.6  501.13  5011.1  505.99
  5040.9  510.32  5135.4  510.82  5174.2  513.43  5218.7  513.29  5224.4   514.3
  5251.2  514.96  5263.1   514.9  5279.7  516.69  5307.6  516.52  5346.4  519.25
    5352  518.17  5368.6  520.03  5374.2  518.76  5390.8  520.47  5396.5  519.76
  5413.1     522  5418.7  521.43  5435.3  523.49  5471.4  523.75  5555.3   527.1
#Mann= 5 ,-1 , 0
  4631.4     .05       0  4908.6      .1       0    4990     .07       0
  5001.6      .1       0  5251.2     .05       0
Bank Sta=4990,5001.6
XS Rating Curve= 0 ,0
Exp/Cntr=0.3,0.1

Type RM Length L Ch R = 1 ,105747  ,721,721,721
BEGIN DESCRIPTION:
Mapping XS f780adec
END DESCRIPTION:
XS GIS Cut Line= 3
      2709337.56      6956496.02      2708832.33      6956092.35
      2708561.46      6955949.11
#Sta/Elev= 30
  4345.9  523.62  4550.2  518.99  4599.9  519.13  4645.7  517.32  4706.3  516.33
    4792  512.15  4812.8  512.69  4841.6  510.23  4905.7  509.62  4920.1  510.43
  4940.9  509.92  4948.9  508.19  4955.3  508.87  4962.3   507.7  4976.1  508.61
  4999.7  506.04  5005.6  500.12  5007.2  499.62  5017.2  500.12  5022.1  506.17
  5027.8  503.74  5044.1  507.62  5050.4     508  5066.2  507.92  5101.6   511.4
  5248.6  518.99  5271.2  521.02  5286.2  523.69  5293.6  526.89    5299  526.89
#Mann= 5 ,-1 , 0
  4345.9     .05       0  4645.7      .1       0  5005.6     .07       0
  5017.2      .1       0  5050.4     .12       0
Bank Sta=5005.6,5017.2
XS Rating Curve= 0 ,0
Exp/Cntr=0.3,0.1

Type RM Length L Ch R = 1 ,105026  ,352,352,352
BEGIN DESCRIPTION:
Mapping XS 12310974
END DESCRIPTION:
XS GIS Cut Line= 3
      2709587.94      6956133.34      2709008.11       6955629.9
      2708213.01      6955539.62
#Sta/Elev= 30
  4231.1  522.27  4255.5  521.54  4319.2  522.39  4509.9  519.28  4542.1  517.49
  4588.9  515.33  4609.7  516.31  4722.3  511.46  4801.6  507.76  4843.3  509.38
  4922.2  507.83  4935.6  509.11  5002.6  508.39  5011.2  507.41  5024.1  499.13
  5025.7  498.63  5035.7  499.13  5041.4  503.74  5051.4  507.21  5061.5  508.55
  5207.4  516.01  5262.8   516.7  5298.7   518.5  5303.8  519.82  5343.3  519.72
  5427.7  524.32    5478  524.36    5515  525.89  5725.7  530.34  5799.2  533.24
#Mann= 8 ,-1 , 0
  4231.1     .05       0  4509.9      .1       0  4542.1     .12       0
  4722.3      .1       0  5024.1     .07       0  5035.7      .1       0
  5427.7     .12       0    5515     .05       0
Bank Sta=5024.1,5035.7
XS Rating Curve= 0 ,0
Exp/Cntr=0.3,0.1

Type RM Length L Ch R = 1 ,104674  ,414,414,414
BEGIN DESCRIPTION:
Mapping XS 782ccfca
END DESCRIPTION:
XS GIS Cut Line= 3
      2709761.58      6955913.58       2709296.3      6955354.55
      2708485.35      6955486.24
#Sta/Elev= 30
  4100.1  520.44  4256.1  518.91  4397.1  518.05  4454.4   519.7  4489.5  518.41
  4506.8  519.27  4524.7  520.48  4663.7  518.02  4688.7  518.53  4730.4  516.14
  4830.1  513.96  4878.4  511.17  4918.9  506.73  4962.9  508.13  4973.9  498.72
  4975.5  498.22  4985.5  498.72  4989.8  504.05  5010.1  508.25  5019.4  508.83
  5060.7  507.18    5162  507.89  5209.2  510.31  5214.3  509.64  5324.1  515.47
  5538.5  522.36  5577.4   523.8  5583.8  522.61  5628.1  525.05    5649  525.14
#Mann= 7 ,-1 , 0
  4100.1     .05       0  4256.1     .12       0  4506.8      .1       0
  4663.7     .12       0  4973.9     .07       0  4985.5     .12       0
  5538.5     .05       0
Bank Sta=4973.9,4985.5
XS Rating Curve= 0 ,0
Exp/Cntr=0.3,0.1

Type RM Length L Ch R = 1 ,104260  ,276,276,276
BEGIN DESCRIPTION:
Mapping XS ec5f540b
END DESCRIPTION:
XS GIS Cut Line= 3
      2709688.68      6955208.72      2708962.97      6955017.75
      2708376.15      6955170.53
#Sta/Elev= 30
  4263.9  518.37  4396.2  515.23  4494.2  515.08  4525.2  513.92  4585.5  514.73
  4625.8  514.01    4631  513.03  4659.5  513.69  4746.8  512.25    4782  508.97
  4787.1  509.41  4804.4  505.73  4814.7  505.38  4887.1  507.67  4949.1  506.94
  4978.4  508.27  5000.8  505.29  5010.2  499.91  5015.7  499.31  5017.3  498.81
  5027.3  499.31  5031.9  507.64  5114.5  506.74  5128.2  507.85  5238.5  510.68
  5354.5  516.98  5447.2  521.12  5482.5  524.36  5538.2  523.52  5620.7  528.27
#Mann= 6 ,-1 , 0
  4263.9     .12       0  4396.2      .1       0  4659.5     .12       0
  5015.7     .07       0  5027.3     .12       0  5354.5     .05       0
Bank Sta=5015.7,5027.3
XS Rating Curve= 0 ,0
Exp/Cntr=0.3,0.1

Type RM Length L Ch R = 1 ,103984  ,332,332,332
BEGIN DESCRIPTION:
Mapping XS d5e04f30
END DESCRIPTION:
XS GIS Cut Line= 4
      2709765.05      6955128.86      2709140.05      6954809.41
      2708935.19        6954799.      2708532.88      6954896.11
#Sta/Elev= 30
  4096.1  517.92  4117.5   517.9  4162.4  514.99  4212.6  516.82  4263.5   513.8
  4321.2  512.94  4353.3  513.93  4385.2   512.4  4473.6  511.37  4679.1  506.09
  4784.6   507.5  4861.2  505.56  4922.2  507.45  4982.3  506.58  5005.3  503.96
    5017  498.18  5018.7  497.68  5028.7  498.18  5030.5  504.56  5035.6  500.48
  5043.4  507.25  5119.4  504.28    5136  506.71  5166.9   508.4  5203.2  508.83
  5228.6  512.12  5348.3  517.54  5375.9  519.31  5382.9   521.2    5417  522.28
#Mann= 6 ,-1 , 0
  4096.1     .12       0  4321.2      .1       0  4385.2     .12       0
    5017     .07       0  5028.7     .12       0  5348.3     .05       0
Bank Sta=5017,5028.7
XS Rating Curve= 0 ,0
Exp/Cntr=0.3,0.1

Type RM Length L Ch R = 1 ,103652  ,665,665,665
BEGIN DESCRIPTION:
Mapping XS a38d3d43
END DESCRIPTION:
XS GIS Cut Line= 3
       2709824.1      6955083.73      2709101.86      6954545.52
      2708501.13      6954493.44
#Sta/Elev= 30
  4022.7  516.19  4081.1  514.84  4122.8  515.75  4166.6  513.75    4235  513.22
  4308.4  513.22  4320.3  512.13  4481.5  506.37  4573.2  505.16  4702.5  505.12
  4767.2  505.92  4781.1  506.85  4808.9  505.66  4917.3  506.82    4923  505.97
  4989.5  505.83  4999.6  503.36  5009.6   498.8  5015.4  497.71  5025.5  498.21
  5029.2  502.82  5034.2  501.45  5039.7  505.97  5180.2  506.03  5300.7  512.57
  5340.8  515.62  5380.2  516.73  5431.2  519.45  5481.4   519.4  5526.4  522.11
#Mann= 6 ,-1 , 0
  4022.7     .12       0    4235     .05       0  4320.3     .12       0
  4989.5     .07       0  5039.7     .12       0  5380.2     .05       0
Bank Sta=4989.5,5039.7
XS Rating Curve= 0 ,0
Exp/Cntr=0.3,0.1
