HEC-RAS study Clear Creek.prj: Clear Creek Base Level Engineering

--- Clear Creek.g01 (geometry) --- (continued)

Type RM Length L Ch R = 1,76436,1041,1041,1041
BEGIN DESCRIPTION:
Clear Creek 121.0
END DESCRIPTION:
XS GIS Cut Line= 3
      2767513.65      6804127.04      2766926.20      6804237.28
      2766350.95      6804339.15
#Sta/Elev= 30
  4402.3  425.12  4411.0  424.04  4546.3  417.36  4603.4  415.47  4616.1  416.03
  4674.6  412.72  4778.8  410.13  4898.5  408.44  4936.4  409.24  4949.3  407.80
  4979.9  409.09  4989.0  408.05  4994.1  405.26  4997.6  400.35  5004.1  400.13
  5005.9  399.63  5016.7  400.13  5030.7  405.84  5040.8  407.79  5061.1  407.37
  5107.1  411.25  5161.2  413.42  5274.4  412.74  5392.6  415.69  5487.7  420.42
  5505.9  423.12  5510.9  422.56  5565.0  426.86  5570.1  425.74  5584.2  427.36
#Mann=5,-1,0
  4402.3    0.05       0  4411.0     0.1       0  4546.3    0.05       0
  5004.1    0.04       0  5016.7    0.05       0
Bank Sta=5004.1,5016.7
Exp/Cntr=0.3,0.1

Type RM Length L Ch R = 1,75395,426,426,426
BEGIN DESCRIPTION:
Clear Creek 120.0
END DESCRIPTION:
XS GIS Cut Line= 3
      2767376.02      6803060.98      2766776.00      6803511.00
      2765876.00      6804111.00
#Sta/Elev= 30
  4242.0  449.24  4313.9  445.16  4392.0  436.31  4434.7  432.79  4442.0  431.88
  4449.3  429.80  4484.7  427.91  4492.0  425.92  4599.3  416.03  4634.7  415.24
  4849.3  406.55  4955.6  404.63  4988.9  406.05  4999.5  405.25  5005.6  405.95
  5014.3  397.02  5016.0  396.52  5026.9  397.02  5028.1  398.21  5035.6  400.07
  5041.6  403.05  5056.6  406.23  5136.3  405.30  5257.9  406.02  5396.2  405.53
  5468.3  406.54  5504.3  407.86  5684.6  420.25  5922.0  430.48  6073.7  439.33
#Mann=3,-1,0
  4242.0    0.05       0  5014.3    0.04       0  5026.9    0.05       0
Bank Sta=5014.3,5026.9
Exp/Cntr=0.3,0.1

Type RM Length L Ch R = 1,74969,440,440,440
BEGIN DESCRIPTION:
Clear Creek 119.0
END DESCRIPTION:
XS GIS Cut Line= 3
      2767176.02      6802860.99      2766576.00      6803211.00
      2766025.99      6803811.01
#Sta/Elev= 30
  4305.3  445.65  4328.5  444.38  4460.4  430.48  4495.1  428.03  4525.3  424.45
  4575.3  421.29  4655.5  413.64  4722.1  409.02  4825.9  404.66  4913.7  403.60
  4964.8  403.53  4986.3  401.65  4992.1  402.94  5007.0  403.55  5016.1  401.08
  5021.2  400.41  5029.1  396.39  5030.9  395.89  5041.7  396.39  5042.2  398.67
  5049.6  400.52  5056.4  403.96  5063.8  404.42  5176.6  402.90  5269.1  404.11
  5516.4  402.81  5629.8  410.01  5686.6  415.52  5778.4  421.81  5813.9  425.58
#Mann=6,-1,0
  4305.3    0.12       0  4460.4    0.05       0  4913.7    0.12       0
  5016.1    0.05       0  5029.1    0.07       0  5041.7    0.05       0
Bank Sta=5029.1,5041.7
Exp/Cntr=0.3,0.1

Type RM Length L Ch R = 1,74529,715,715,715
BEGIN DESCRIPTION:
Clear Creek 118.0
END DESCRIPTION:
XS GIS Cut Line= 3
      2766925.99      6802661.00      2766526.00      6802811.00
      2765326.03      6803410.98
#Sta/Elev= 30
  4565.8  434.82  4587.4  432.77  4676.1  424.20  4746.5  416.60  4864.1  406.66
  4892.4  403.91  4928.9  402.18  5037.7  398.96  5046.1  399.91  5060.1  395.31
  5067.8  395.08  5069.5  394.58  5080.4  395.08  5081.6  396.44  5090.8  402.61
  5240.4  401.03  5538.0  399.98  5784.0  400.56  5923.8  403.38  5976.9  402.91
  6013.2  403.78  6102.6  408.83  6164.1  414.65  6169.7  414.23  6192.1  416.19
  6208.9  418.94  6236.8  420.82  6253.6  423.62  6312.3  430.24  6334.6  430.46
#Mann=8,-1,0
  4565.8    0.12       0  4587.4     0.1       0  4676.1    0.12       0
  4864.1     0.1       0  5067.8    0.07       0  5080.4     0.1       0
  5081.6    0.12       0  5240.4    0.05       0
Bank Sta=5067.8,5080.4
Exp/Cntr=0.3,0.1

Type RM Length L Ch R = 1,73814,617,617,617
BEGIN DESCRIPTION:
Clear Creek 117.0
END DESCRIPTION:
XS GIS Cut Line= 3
      2767076.01      6802411.00      2765981.99      6802612.96
      2765242.58      6803116.70
#Sta/Elev= 30
  3887.5  436.91  3928.2  436.18  4019.7  429.02  4025.0  422.79  4050.2  420.42
  4078.0  420.33  4090.9  426.12  4119.5  425.00  4182.4  418.13  4300.0  408.83
  4426.5  402.13  4558.7  399.63  4680.7  401.35  4850.0  398.59  4961.0  400.48
  4975.6  398.72  4989.1  394.28  4990.9  393.78  5001.7  394.28  5003.3  399.08
  5012.4  398.97  5030.0  400.57  5151.8  399.40  5168.7  398.95  5297.7  398.64
  5470.2  401.92  5506.1  404.65  5586.8  417.64  5628.7  420.85  5894.7  433.05
#Mann=8,-1,0
  3887.5    0.12       0  4119.5    0.05       0  4989.1    0.04       0
  5001.7    0.05       0  5012.4    0.12       0  5030.0    0.05       0
  5151.8    0.12       0  5168.7    0.05       0
Bank Sta=4989.1,5001.7
Exp/Cntr=0.3,0.1

Type RM Length L Ch R = 1,73197,929,929,929
BEGIN DESCRIPTION:
Clear Creek 116.0
END DESCRIPTION:
XS GIS Cut Line= 3
      2767325.97      6802011.01      2765526.00      6802311.00
      2765176.01      6802910.99
#Sta/Elev= 30
  3174.5  445.89  3296.1  435.93  3458.3  425.51  3671.2  414.66  3681.4  413.52
  3689.0  410.06  3694.0  409.42  3711.8  412.86  3721.9  410.44  3876.5  408.70
  3932.3  405.13  3998.2  404.74  4218.7  398.11  4723.0  396.51  4989.2  398.82
  4996.8  393.16  4999.3  393.16  5000.8  391.13  5002.6  390.63  5013.5  391.13
  5022.4  398.26  5028.7  398.87  5050.2  398.03  5093.2  401.05  5167.6  403.50
  5386.7  407.45  5627.3  418.98  5664.6  421.72  5686.1  426.34  5693.9  426.28
#Mann=3,-1,0
  3174.5    0.05       0  5000.8    0.04       0  5013.5    0.05       0
Bank Sta=5000.8,5013.5
Exp/Cntr=0.3,0.1

Type RM Length L Ch R = 1,72268,414,414,414
BEGIN DESCRIPTION:
Clear Creek 115.0
END DESCRIPTION:
XS GIS Cut Line= 3
      2765546.18      6799578.06      2765176.00      6801611.00
      2765082.37      6802891.81
#Sta/Elev= 30
  2944.0  437.88  3142.8  425.51  3394.2  404.39  3497.1  400.10  3648.3  396.19
  3841.5  397.48  3851.6  392.61  3861.4  391.87  3866.5  393.68  3872.0  391.83
  3892.3  397.37  4024.6  394.74  4805.2  393.65  4978.6  395.14  5001.5  389.31
  5003.2  388.81  5014.2  389.31  5040.5  395.39  5077.3  392.91  5082.3  395.44
  5160.8  395.20  5170.8  389.53  5190.9  392.19  5200.9  389.85  5210.9  391.02
  5217.2  395.67  5692.2  396.66  6193.5  420.64  6223.6  425.20  6294.6  424.34
#Mann=7,-1,0
  2944.0     0.1       0  3497.1    0.12       0  4024.6    0.05       0
  4805.2    0.12       0  5001.5    0.07       0  5014.2    0.12       0
  5217.2    0.05       0
Bank Sta=5001.5,5014.2
Exp/Cntr=0.3,0.1

Type RM Length L Ch R = 1,71854,446,446,446
BEGIN DESCRIPTION:
Clear Creek 114.0
END DESCRIPTION:
XS GIS Cut Line= 3
      2765011.74      6799537.23      2764876.00      6801361.00
      2764970.82      6802882.13
#Sta/Elev= 30
  3176.1  438.07  3200.1  438.56  3266.7  436.13  3323.0  433.59  3370.4  429.02
  3390.5  425.14  3571.0  412.53  3911.9  399.91  4072.3  395.60  4353.1  394.18
  4383.2  390.95  4398.4  394.57  4663.5  391.46  4938.6  393.83  4944.7  393.72
  4958.5  388.86  4960.2  388.36  4971.2  388.86  4974.8  392.63  4984.9  393.76
  5161.1  392.31  5259.4  392.18  5436.0  393.99  5546.0  393.50  5676.2  398.14
  5890.3  399.69  6016.9  406.97  6206.3  412.48  6366.8  424.69  6529.0  428.38
#Mann=8,-1,0
  3176.1    0.05       0  3200.1    0.12       0  3266.7    0.05       0
  4958.5    0.07       0  4971.2    0.05       0  5161.1    0.05       0
  5259.4    0.12       0  5436.0    0.05       0
Bank Sta=4958.5,4971.2
Exp/Cntr=0.3,0.1

Type RM Length L Ch R = 1,71408,912,912,912
BEGIN DESCRIPTION:
Clear Creek 113.0
END DESCRIPTION:
XS GIS Cut Line= 3
      2764775.99      6799511.04      2764476.00      6801311.00
      2764859.46      6802825.22
#Sta/Elev= 30
  3174.5  458.54  3219.5  456.33  3312.4  448.78  3478.6  432.96  3615.1  414.84
  3810.6  400.20  4109.6  393.45  4391.0  392.59  4406.3  389.91  4411.3  387.77
  4431.6  393.09  4634.3  390.96  4654.6  387.84  4662.2  390.55  4929.3  391.36
  4989.1  392.61  4990.4  387.42  4992.2  386.92  5003.2  387.42  5009.6  387.61
  5017.2  392.34  5022.4  388.22  5030.2  392.87  5058.2  394.19  5339.7  391.62
  5979.3  395.12  6113.4  398.52  6318.9  407.40  6453.8  420.81  6561.3  427.96
#Mann=9,-1,0
  3174.5    0.12       0  3219.5    0.05       0  3312.4    0.12       0
  3615.1    0.05       0  4109.6     0.1       0  4406.3    0.05       0
  4929.3    0.12       0  4990.4    0.05       0  5003.2    0.05       0
Bank Sta=4990.4,5003.2
Exp/Cntr=0.3,0.1

Type RM Length L Ch R = 1,70496,468,468,468
BEGIN DESCRIPTION:
Clear Creek 112.0
END DESCRIPTION:
XS GIS Cut Line= 4
      2763895.86      6799892.11      2763926.00      6800761.00
      2764134.50      6802248.05      2764765.54      6802886.52
#Sta/Elev= 30
  4130.9  424.99  4189.8  422.98  4269.9  417.83  4289.9  415.44  4465.6  403.06
  4566.3  397.53  4700.1  395.93  4780.2  393.38  4960.3  390.25  4990.3  390.43
  4997.8  386.86  5002.6  385.85  5004.6  385.35  5018.2  385.85  5020.5  390.88
  5154.1  389.97  5424.4  389.38  5683.2  391.83  5798.0  391.63  5989.9  394.74
  6121.4  394.56  6500.9  398.33  6929.3  397.00  7028.3  398.20  7077.8  398.95
  7169.7  402.30  7275.8  407.91  7297.0  410.53  7346.5  414.40  7399.6  423.00
#Mann=5,-1,0
  4130.9    0.05       0  4465.6    0.12       0  5002.6    0.07       0
  5018.2    0.12       0  5154.1    0.05       0
Bank Sta=5002.6,5018.2
Exp/Cntr=0.3,0.1

Type RM Length L Ch R = 1,70028,435,435,435
BEGIN DESCRIPTION:
Clear Creek 111.0
END DESCRIPTION:
XS GIS Cut Line= 3
      2763576.00      6800111.04      2763526.00      6800661.00
      2763644.29      6802467.91
#Sta/Elev= 30
  4452.7  439.25  4553.1  418.18  4603.3  409.58  4663.5  400.87  4693.6  397.46
  4784.0  390.20  4864.3  389.03  4924.6  390.25  4926.8  384.11  4928.8  383.61
  4942.4  384.11  4954.7  386.37  4964.8  390.18  5306.8  388.19  5967.0  391.18
  6037.1  393.00  6097.3  393.22  6157.7  396.37  6167.4  394.96  6187.5  388.33
  6207.5  393.36  6227.5  395.49  6287.7  394.43  6309.4  395.61  6397.9  405.97
  6438.0  412.21  6538.2  421.81  6612.8  422.62  6728.6  421.51  6815.7  423.12
#Mann=4,-1,0
  4452.7    0.12       0  4926.8    0.07       0  4942.4    0.12       0
  5306.8    0.05       0
Bank Sta=4926.8,4942.4
Exp/Cntr=0.3,0.1

Type RM Length L Ch R = 1,69593,472,472,472
BEGIN DESCRIPTION:
Clear Creek 110.0
END DESCRIPTION:
XS GIS Cut Line= 3
      2762820.69      6800309.15      2763126.00      6800761.00
      2763478.09      6802535.07
#Sta/Elev= 30
  4458.9  419.67  4478.3  417.06  4529.2  414.72  4787.0  395.25  4810.9  392.15
  4873.9  388.75  4882.8  390.35  4924.8  386.71  4960.8  387.35  4967.9  381.95
  4969.9  381.45  4983.6  381.95  4996.7  383.48  5001.2  389.22  5167.3  386.37
  5367.9  387.43  5666.9  389.59  5830.0  393.15  5848.6  388.53  5853.7  390.34
  5860.6  387.57  5881.0  387.39  5932.0  393.65  5972.8  392.81  6053.3  396.78
  6109.5  397.16  6365.4  409.60  6543.7  413.82  6723.6  422.45  6812.9  423.17
#Mann=4,-1,0
  4458.9    0.12       0  4967.9    0.07       0  4983.6    0.12       0
  5367.9    0.05       0
Bank Sta=4967.9,4983.6
Exp/Cntr=0.3,0.1

Type RM Length L Ch R = 1,69121,303,303,303
BEGIN DESCRIPTION:
Clear Creek 109.0
END DESCRIPTION:
XS GIS Cut Line= 3
      2762726.00      6800511.00      2762776.00      6800961.00
      2763074.38      6802676.78
#Sta/Elev= 30
  4536.6  420.97  4858.6  388.86  4939.1  388.62  4961.3  380.53  4963.3  380.03
  4977.1  380.53  4991.9  382.71  4999.5  387.01  5009.7  386.85  5021.7  380.61
  5030.0  382.04  5040.1  387.71  5114.6  386.74  5243.1  386.48  5385.5  389.93
  5405.5  388.97  5415.7  383.01  5423.9  387.93  5429.0  387.09  5436.0  390.41
  5504.9  389.51  5537.5  388.73  5567.9  391.01  5604.8  389.06  5689.6  389.07
  5852.1  402.25  6069.8  403.23  6379.9  414.50  6572.8  425.70  6730.9  426.52
#Mann=8,-1,0
  4536.6    0.12       0  4961.3    0.07       0  4977.1    0.12       0
  5114.6    0.05       0  5385.5    0.12       0  5504.9    0.05       0
  5604.8    0.12       0  5689.6    0.05       0
Bank Sta=4961.3,4977.1
Exp/Cntr=0.3,0.1

Type RM Length L Ch R = 1,68818,1069,1069,1069
BEGIN DESCRIPTION:
Clear Creek 108.0
END DESCRIPTION:
XS GIS Cut Line= 3
      2762526.00      6800610.98      2762519.94      6801058.44
      2762802.65      6802726.14
#Sta/Elev= 30
  4552.5  402.61  4672.5  396.08  4742.5  390.64  4812.5  387.59  4982.6  386.84
  4990.9  379.58  4992.9  379.08  5006.7  379.58  5012.7  387.44  5164.9  384.58
  5364.0  388.40  5369.1  387.93  5377.9  381.35  5388.0  383.14  5398.2  387.52
  5408.3  388.59  5519.9  387.24  5611.2  390.29  5721.0  399.32  5854.6  401.61
  5885.0  400.02  5895.8  401.28  6067.6  403.67  6083.1  405.53  6250.1  410.92
  6351.6  416.90  6402.3  417.55  6445.1  420.25  6574.7  423.00  6691.5  423.43
#Mann=4,-1,0
  4552.5    0.12       0  4990.9    0.07       0  5006.7    0.12       0
  5895.8    0.05       0
Bank Sta=4990.9,5006.7
Exp/Cntr=0.3,0.1

Type RM Length L Ch R = 1,67749,532,532,532
BEGIN DESCRIPTION:
Clear Creek 107.0
END DESCRIPTION:
XS GIS Cut Line= 3
      2761458.81      6799847.19      2762026.00      6801611.00
      2762554.99      6802807.73
#Sta/Elev= 30
  3148.1  427.71  3546.6  417.15  3803.3  413.86  3845.9  414.74  3872.8  412.79
  3937.1  413.64  3950.4  414.89  3969.0  412.44  3974.3  413.61  4087.0  397.54
  4231.0  386.21  4357.1  385.55  4805.8  384.85  4843.3  383.63  4895.8  385.37
  4920.6  382.77  4979.6  386.68  4990.4  386.04  4998.2  378.31  5006.1  377.78
  5008.1  377.28  5024.3  377.78  5033.1  385.14  5146.5  392.75  5288.0  399.18
  5525.7  400.24  5874.5  406.27  5984.9  411.78  6100.6  413.77  6309.3  421.17
#Mann=7,-1,0
  3148.1    0.05       0  3937.1    0.12       0  4357.1    0.05       0
  4805.8    0.12       0  5006.1    0.07       0  5024.3    0.12       0
  5146.5    0.05       0
Bank Sta=5006.1,5024.3
Exp/Cntr=0.3,0.1

Type RM Length L Ch R = 1,67217,545,545,545
BEGIN DESCRIPTION:
Clear Creek 106.0
END DESCRIPTION:
XS GIS Cut Line= 3
      2761095.50      6799966.47      2761576.00      6801761.00
      2761664.38      6802931.42
#Sta/Elev= 30
  3146.5  424.38  3362.2  418.19  3592.1  401.27  3747.1  396.09  3752.3  397.46
  3756.9  395.09  3762.0  392.46  3787.1  397.23  3851.9  394.30  4062.2  388.84
  4131.9  385.60  4283.4  383.12  4421.9  383.53  4676.9  382.61  4693.7  383.88
  4939.1  385.41  4962.8  385.23  4964.1  376.38  4966.1  375.88  4982.3  376.38
  4993.9  385.52  5054.4  383.77  5070.0  386.74  5164.7  391.44  5219.5  396.47
  5265.0  398.71  5338.2  398.32  5595.9  401.83  5977.0  415.30  6178.0  417.99
#Mann=9,-1,0
  3146.5    0.05       0  3756.9    0.12       0  3851.9    0.05       0
  4283.4    0.12       0  4421.9    0.05       0  4939.1    0.12       0
  4964.1    0.07       0  4982.3    0.12       0  5219.5    0.05       0
Bank Sta=4964.1,4982.3
Exp/Cntr=0.3,0.1

Type RM Length L Ch R = 1,66672,568,568,568
BEGIN DESCRIPTION:
Clear Creek 105.0
END DESCRIPTION:
XS GIS Cut Line= 3
      2760682.31      6800425.30      2761126.00      6801761.00
      2761298.71      6802466.29
#Sta/Elev= 30
  3592.2  420.31  3648.6  423.67  3735.2  426.35  3791.1  422.72  3834.7  418.34
  3945.9  405.47  4051.3  395.73  4127.7  390.44  4229.6  383.91  4293.7  380.90
  4462.3  379.46  4515.0  380.81  4693.6  380.70  4848.3  383.61  4920.5  383.10
  4957.5  384.32  4968.1  378.22  4969.5  375.23  4971.5  374.73  4987.7  375.23
  4997.0  381.60  5002.2  381.60  5010.0  383.65  5030.6  382.82  5054.9  387.67
  5215.9  398.67  5257.1  399.65  5527.5  397.66  5605.6  398.50  5725.8  402.00
#Mann=9,-1,0
  3592.2    0.05       0  3791.1    0.12       0  3834.7     0.1       0
  4127.7    0.12       0  4229.6    0.05       0  4848.3    0.12       0
  4969.5    0.07       0  4987.7    0.12       0  5054.9    0.05       0
Bank Sta=4969.5,4987.7
Exp/Cntr=0.3,0.1

Type RM Length L Ch R = 1,66104,521,521,521
BEGIN DESCRIPTION:
Clear Creek 104.0
END DESCRIPTION:
XS GIS Cut Line= 3
      2760240.88      6800749.16      2760626.00      6801661.00
      2760815.69      6802371.58
#Sta/Elev= 30
  4005.4  442.78  4040.0  437.88  4104.1  431.04  4156.9  423.31  4238.9  414.74
  4286.3  407.63  4291.7  408.63  4404.2  399.42  4421.1  399.26  4430.8  397.17
  4511.6  390.38  4645.3  381.04  4734.9  378.82  4919.2  380.06  4997.8  382.35
  5003.6  374.41  5005.6  373.91  5021.8  374.41  5026.3  379.24  5036.6  382.65
  5107.7  382.77  5160.8  381.26  5266.6  380.53  5328.2  380.67  5409.2  388.76
  5489.1  392.13  5585.2  393.90  5633.4  397.43  5668.0  398.23  5730.7  396.18
#Mann=9,-1,0
  4005.4     0.1       0  4404.2    0.12       0  4511.6    0.05       0
  4734.9    0.12       0  5003.6    0.07       0  5021.8    0.12       0
  5107.7    0.05       0  5266.6    0.12       0  5489.1    0.05       0
Bank Sta=5003.6,5021.8
Exp/Cntr=0.3,0.1

Type RM Length L Ch R = 1,65583,553,553,553
BEGIN DESCRIPTION:
Clear Creek 103.0
END DESCRIPTION:
XS GIS Cut Line= 3
      2760126.00      6800761.00      2760226.00      6801561.00
      2760343.90      6802536.37
#Sta/Elev= 30
  4189.1  449.18  4239.5  441.01  4388.1  422.96  4549.4  404.91  4577.7  402.85
  4602.3  401.60  4642.6  396.12  4662.8  395.71  4753.5  386.31  4839.0  380.79
  4934.9  377.94  4975.2  379.46  4985.3  381.09  4997.8  378.84  5006.3  373.51
  5008.3  373.01  5024.6  373.51  5025.5  376.44  5033.8  381.63  5036.9  379.27
  5038.8  377.82  5045.7  381.70  5109.7  380.52  5135.8  380.10  5509.0  378.29
  5680.3  377.78  5731.8  381.45  5881.7  394.13  5950.4  394.32  5977.8  393.01
#Mann=10,-1,0
  4189.1     0.1       0  4577.7    0.05       0  4839.0    0.12       0
  5006.3    0.07       0  5024.6    0.12       0  5036.9    0.05       0
  5109.7    0.12       0  5135.8    0.05       0  5509.0    0.12       0
  5731.8    0.05       0
Bank Sta=5006.3,5024.6
Exp/Cntr=0.3,0.1

Type RM Length L Ch R = 1,65030,574,574,574
BEGIN DESCRIPTION:
Clear Creek 102.0
END DESCRIPTION:
XS GIS Cut Line= 3
      2759783.24      6800696.46      2759776.00      6801711.00
      2759811.04      6802565.01
#Sta/Elev= 30
  3989.7  426.66  4054.2  425.07  4114.2  421.23  4314.3  404.41  4434.3  397.30
  4484.3  392.25  4553.7  389.58  4584.3  388.19  4614.3  384.72  4784.3  378.99
  4934.3  380.38  4984.3  380.02  4992.6  372.49  4994.6  371.99  5010.9  372.49
  5014.3  377.96  5024.3  380.69  5178.9  378.78  5234.5  377.98  5314.5  379.36
  5324.5  378.33  5354.6  379.36  5375.1  378.97  5473.2  377.63  5581.6  377.42
  5611.9  376.63  5674.8  377.12  5734.9  381.07  5804.9  387.54  5859.0  389.56
#Mann=8,-1,0
  3989.7     0.1       0  4553.7    0.05       0  4992.6    0.04       0
  5010.9    0.05       0  5178.9    0.12       0  5375.1    0.05       0
  5473.2    0.12       0  5581.6    0.05       0
Bank Sta=4992.6,5010.9
Exp/Cntr=0.3,0.1

Type RM Length L Ch R = 1,64456,677,677,677
BEGIN DESCRIPTION:
Clear Creek 101.0
END DESCRIPTION:
XS GIS Cut Line= 3
      2759355.27      6800466.98      2759326.00      6801761.00
      2759685.39      6802566.73
#Sta/Elev= 30
  3722.8  439.50  3911.8  422.89  3996.9  414.44  4146.9  403.53  4226.9  399.60
  4427.0  395.92  4597.0  383.55  4777.1  378.51  4847.1  377.47  4875.7  378.33
  4887.1  375.94  4897.1  378.44  4937.1  378.47  4947.1  373.34  4957.1  370.09
  4967.9  369.84  4969.9  369.34  4986.3  369.84  4987.1  371.17  4997.1  378.39
  5012.9  378.81  5083.4  378.21  5129.9  377.15  5147.6  375.75  5235.6  376.28
  5481.2  376.78  5720.1  376.89  5766.5  379.19  5813.0  382.83  5899.4  386.73
#Mann=7,-1,0
  3722.8    0.05       0  4875.7    0.12       0  4967.9    0.07       0
  4986.3    0.12       0  5012.9    0.05       0  5235.6    0.12       0
  5481.2    0.05       0
Bank Sta=4967.9,4986.3
Exp/Cntr=0.3,0.1

Type RM Length L Ch R = 1,63779,415,415,415
BEGIN DESCRIPTION:
Mapping XS e212a9bd
END DESCRIPTION:
XS GIS Cut Line= 3
      2758890.45      6800738.87      2758862.63      6801881.16
      2758985.34      6803423.25
#Sta/Elev= 30
  3863.6  410.81  3975.8  403.20  3985.8  401.46  4015.8  399.32  4035.8  395.41
  4095.8  393.04  4135.8  393.13  4345.9  383.19  4636.0  376.51  4726.0  375.90
  4776.0  377.44  4946.1  377.05  4966.1  368.77  5006.6  368.21  5008.6  367.71
  5025.6  368.21  5036.2  368.57  5046.2  370.18  5056.2  375.55  5066.3  377.10
  5126.4  376.80  5266.9  373.68  5447.5  375.40  5818.6  376.38  6049.4  381.04
  6245.7  388.87  6320.2  389.98  6350.3  389.36  6480.7  392.23  6553.2  391.42
#Mann=3,-1,0
  3863.6    0.05       0  5006.6    0.04       0  5025.6    0.05       0
Bank Sta=5006.6,5025.6
Exp/Cntr=0.3,0.1

Type RM Length L Ch R = 1,63364,529,529,529
BEGIN DESCRIPTION:
Clear Creek 100.0
END DESCRIPTION:
XS GIS Cut Line= 3
      2758704.27      6800018.23      2758476.00      6801961.00
      2758714.84      6803097.85
#Sta/Elev= 30
  3043.5  442.01  3187.2  435.86  3318.1  428.05  3325.9  427.35  3330.9  425.12
  3348.3  427.02  3579.9  423.54  3839.7  412.37  3952.5  409.13  4270.4  384.59
  4365.3  379.58  4596.9  375.08  4858.7  373.59  4898.9  375.82  4969.4  375.92
  5002.2  373.29  5010.0  367.51  5012.0  367.01  5029.0  367.51  5030.3  371.76
  5040.5  375.87  5306.2  371.03  5357.3  371.17  5377.7  372.82  5490.1  372.27
  5602.5  376.32  5633.2  379.81  5674.0  381.61  5960.1  387.83  6161.3  389.18
#Mann=3,-1,0
  3043.5    0.05       0  5010.0    0.04       0  5029.0    0.05       0
Bank Sta=5010,5029
Exp/Cntr=0.3,0.1

Type RM Length L Ch R = 1,62835,901,901,901
BEGIN DESCRIPTION:
Clear Creek 99.0
END DESCRIPTION:
XS GIS Cut Line= 3
      2757996.28      6800702.38      2758076.00      6801961.00
      2758324.64      6803012.25
#Sta/Elev= 30
  3739.3  421.19  3788.0  419.55  3838.1  415.99  3918.3  412.86  4068.6  401.59
  4148.7  394.47  4168.8  391.67  4228.9  388.68  4349.1  380.00  4409.3  377.22
  4569.6  372.52  4739.9  373.05  4910.3  372.49  4918.3  373.32  4980.4  374.70
  4990.4  373.41  4997.9  366.79  5001.2  366.10  5003.2  365.60  5020.2  366.10
  5024.2  372.76  5041.5  374.56  5319.0  371.33  5709.5  370.61  5781.4  375.08
  5805.7  377.47  5842.8  379.05  5853.3  380.54  5979.9  387.86  6080.7  387.66
#Mann=3,-1,0
  3739.3    0.05       0  5001.2    0.04       0  5020.2    0.05       0
Bank Sta=5001.2,5020.2
Exp/Cntr=0.3,0.1

Type RM Length L Ch R = 1,61934,610,610,610
BEGIN DESCRIPTION:
Mapping XS 6018c6fc
END DESCRIPTION:
XS GIS Cut Line= 3
      2757562.69      6800641.03      2757330.60      6802201.00
      2757881.45      6803481.07
#Sta/Elev= 30
  3459.9  408.25  3574.9  401.69  3661.4  398.50  3743.0  394.92  3815.0  390.43
  3854.2  391.63  3943.6  388.73  3955.3  387.07  4018.0  384.50  4127.1  381.27
  4167.6  377.49  4216.0  375.60  4456.0  371.27  4493.4  369.85  4531.5  371.02
  4580.5  368.98  4996.6  371.43  5006.7  370.96  5023.6  363.35  5025.6  362.85
  5042.6  363.35  5047.9  370.30  5063.8  370.99  5134.4  369.16  5461.6  367.86
  5800.8  369.08  5876.8  372.04  6099.5  385.33  6222.7  390.93  6430.6  396.55
#Mann=8,-1,0
  3459.9    0.05       0  3574.9    0.12       0  3661.4    0.05       0
  3743.0    0.12       0  4456.0    0.05       0  4580.5    0.12       0
  5023.6    0.07       0  5042.6    0.05       0
Bank Sta=5023.6,5042.6
Exp/Cntr=0.3,0.1

Type RM Length L Ch R = 1,61324,1206,1206,1206
BEGIN DESCRIPTION:
Mapping XS 0c433fc2
END DESCRIPTION:
XS GIS Cut Line= 3
      2757431.68      6800660.36      2756858.82      6802140.18
      2757567.56      6803226.38
#Sta/Elev= 30
  3403.1  401.40  3491.5  396.59  3988.8  375.03  4125.2  371.97  4229.2  370.21
  4398.9  368.00  4448.0  368.82  4519.0  367.29  4645.5  368.17  4940.1  368.79
  5002.8  370.03  5010.5  368.84  5016.1  363.17  5018.1  362.67  5035.1  363.17
  5038.7  363.82  5046.7  370.24  5146.2  367.87  5155.4  366.30  5161.3  367.14
  5170.0  364.60  5176.4  367.46  5258.7  367.85  5632.1  370.35  5985.0  370.72
  6057.4  373.57  6129.9  378.37  6238.5  388.21  6268.5  389.02  6286.9  388.06
#Mann=10,-1,0
  3403.1    0.05       0  3988.8    0.12       0  4125.2     0.1       0
  4229.2    0.12       0  4448.0     0.1       0  4645.5    0.12       0
  4940.1     0.1       0  5016.1    0.07       0  5035.1     0.1       0
  5258.7    0.05       0
Bank Sta=5016.1,5035.1
Exp/Cntr=0.3,0.1

Type RM Length L Ch R = 1,60118,522,522,522
BEGIN DESCRIPTION:
Clear Creek 98.0
END DESCRIPTION:
XS GIS Cut Line= 3
      2757426.02      6800360.97      2755876.00      6801961.00
      2755565.02      6803141.53
#Sta/Elev= 30
  2772.0  415.23  2963.0  402.76  3168.1  394.74  3236.5  390.11  3358.9  380.37
  3479.3  375.19  3493.4  373.42  3896.5  367.25  4155.7  365.01  4299.6  366.10
  4491.6  365.10  4558.8  365.51  4637.3  365.50  4936.0  367.81  4950.2  363.06
  4953.3  358.24  4955.5  357.74  4975.3  358.24  4985.7  365.97  4992.6  367.68
  5068.3  371.19  5123.8  373.97  5144.5  376.62  5237.5  379.21  5403.0  390.84
  5630.5  403.25  5781.3  403.30  5840.9  402.56  6074.6  405.00  6220.5  405.04
#Mann=11,-1,0
  2772.0    0.05       0  3236.5    0.12       0  4155.7    0.05       0
  4491.6    0.12       0  4558.8     0.1       0  4637.3    0.12       0
  4953.3    0.07       0  4975.3    0.12       0  5068.3    0.05       0
  5781.3    0.12       0  5840.9    0.05       0
Bank Sta=4953.3,4975.3
Exp/Cntr=0.3,0.1

Type RM Length L Ch R = 1,59596,538,538,538
BEGIN DESCRIPTION:
Clear Creek 97.0
END DESCRIPTION:
XS GIS Cut Line= 3
      2756426.01      6800410.99      2755626.00      6801561.00
      2755576.00      6802011.02
#Sta/Elev= 30
  3599.3  399.29  3627.4  398.02  3628.3  397.94  3721.3  391.15  3757.7  389.28
  3862.4  380.21  4044.9  368.18  4155.7  366.02  4184.9  365.87  4325.1  364.52
  4381.8  361.77  4425.1  362.09  4439.9  364.19  4453.4  364.44  4476.4  363.43
  4641.0  365.27  4756.6  363.83  4918.6  366.08  4986.7  366.30  4992.8  357.23
  4999.3  356.64  5001.5  356.14  5021.3  356.64  5030.2  360.05  5040.5  360.30
  5050.5  366.99  5128.4  366.84  5161.2  365.98  5221.6  366.89  5453.0  382.23
#Mann=13,-1,0
  3599.3    0.12       0  3627.4    0.05       0  3628.3    0.12       0
  3721.3     0.1       0  3862.4    0.05       0  4155.7    0.12       0
  4184.9    0.05       0  4425.1    0.12       0  4918.6     0.1       0
  4999.3    0.07       0  5021.3     0.1       0  5030.2    0.12       0
  5128.4    0.05       0
Bank Sta=4999.3,5021.3
Exp/Cntr=0.3,0.1

Type RM Length L Ch R = 1,59058,751,751,751
BEGIN DESCRIPTION:
Clear Creek 96.0
END DESCRIPTION:
XS GIS Cut Line= 3
      2755909.59      6800153.89      2755276.00      6801461.00
      2755053.03      6802116.02
#Sta/Elev= 30
  3554.2  398.67  3688.4  392.11  3965.7  377.23  4012.5  373.36  4084.4  369.59
  4355.0  363.50  4384.5  361.31  4439.8  362.49  4480.3  360.63  4490.5  362.69
  4513.1  363.24  4602.7  362.64  4770.6  363.68  4826.0  364.22  4917.9  365.71
  4925.0  361.17  4930.5  365.77  4934.9  363.94  4947.6  356.34  4951.3  356.24
  4953.5  355.74  4973.4  356.24  4992.7  365.38  4998.3  363.38  5004.0  365.21
  5143.7  364.85  5273.3  365.32  5367.4  367.74  5607.8  385.72  5698.7  390.57
#Mann=11,-1,0
  3554.2    0.12       0  3688.4     0.1       0  4012.5    0.12       0
  4480.3     0.1       0  4602.7    0.12       0  4770.6     0.1       0
  4826.0    0.12       0  4934.9     0.1       0  4951.3    0.07       0
  4973.4     0.1       0  5143.7    0.05       0
Bank Sta=4951.3,4973.4
Exp/Cntr=0.3,0.1

Type RM Length L Ch R = 1,58307,322,322,322
BEGIN DESCRIPTION:
Clear Creek 95.0
END DESCRIPTION:
XS GIS Cut Line= 3
      2755466.07      6799943.92      2754876.00      6801311.00
      2754676.00      6802011.00
#Sta/Elev= 30
  3675.0  393.83  3968.4  387.13  4109.7  379.16  4227.3  370.96  4324.3  365.85
  4335.6  365.79  4634.2  361.05  4699.1  361.42  4717.2  358.36  4728.3  361.43
  4744.1  361.72  4880.8  361.79  4957.0  364.20  4967.9  359.16  4968.5  354.86
  4970.7  354.36  4990.6  354.86  4997.6  362.73  5034.9  363.80  5088.9  364.16
  5236.8  364.48  5434.7  362.12  5438.9  362.19  5511.1  363.54  5600.8  371.87
  5632.0  373.16  5736.0  385.86  5797.1  390.91  5836.1  396.50  5892.0  401.55
#Mann=12,-1,0
  3675.0     0.1       0  4109.7    0.12       0  4324.3     0.1       0
  4335.6    0.12       0  4634.2     0.1       0  4744.1    0.12       0
  4968.5    0.07       0  4990.6    0.12       0  5034.9     0.1       0
  5088.9    0.12       0  5434.7     0.1       0  5438.9    0.05       0
Bank Sta=4968.5,4990.6
Exp/Cntr=0.3,0.1

Type RM Length L Ch R = 1,57985,561,561,561
BEGIN DESCRIPTION:
Clear Creek 94.0
END DESCRIPTION:
XS GIS Cut Line= 3
      2755326.00      6799911.01      2754676.00      6801061.00
      2754576.00      6801861.00
#Sta/Elev= 30
  3682.9  401.18  3694.4  401.12  3879.9  398.15  4157.1  375.45  4203.3  372.96
  4234.3  369.02  4403.9  363.24  4505.1  361.30  4636.3  361.48  4645.1  360.81
  4659.3  356.83  4666.8  359.52  4672.5  358.31  4688.4  361.57  4753.4  360.87
  4946.4  363.58  4952.6  361.60  4958.4  362.13  4963.2  354.82  4965.4  354.32
  4985.3  354.82  4990.2  359.03  4995.9  358.29  5001.0  362.95  5021.6  362.66
  5316.8  362.38  5477.5  361.39  5526.0  366.36  5691.7  383.57  5810.1  392.72
#Mann=9,-1,0
  3682.9    0.12       0  3694.4     0.1       0  4157.1    0.12       0
  4403.9     0.1       0  4963.2    0.07       0  4985.3     0.1       0
  5021.6    0.12       0  5316.8     0.1       0  5526.0    0.05       0
Bank Sta=4963.2,4985.3
Exp/Cntr=0.3,0.1

Type RM Length L Ch R = 1,57424,541,541,541
BEGIN DESCRIPTION:
Clear Creek 93.0
END DESCRIPTION:
XS GIS Cut Line= 3
      2755125.97      6800061.04      2754376.00      6800861.00
      2754575.99      6802110.96
#Sta/Elev= 30
  3903.3  397.80  4023.6  386.66  4238.0  370.93  4306.5  366.12  4478.7  361.41
  4617.6  360.01  4709.9  361.52  4745.1  359.95  4752.4  357.95  4759.3  358.37
  4766.6  355.95  4773.4  357.16  4780.5  360.31  4964.4  362.26  4967.5  352.81
  4969.7  352.31  4989.6  352.81  4992.8  353.96  4996.4  360.66  5010.0  361.01
  5111.2  362.68  5637.9  360.46  5732.1  369.90  5830.3  378.85  5880.9  385.94
  5917.0  389.43  5922.0  388.48  5984.1  391.80  6093.6  399.86  6265.7  399.78
#Mann=6,-1,0
  3903.3     0.1       0  4238.0    0.12       0  4478.7     0.1       0
  4967.5    0.07       0  4989.6     0.1       0  5732.1    0.05       0
Bank Sta=4967.5,4989.6
Exp/Cntr=0.3,0.1

Type RM Length L Ch R = 1,56883,575,575,575
BEGIN DESCRIPTION:
Clear Creek 92.0
END DESCRIPTION:
XS GIS Cut Line= 3
      2754875.96      6799961.03      2754076.00      6800611.00
      2754426.00      6802010.98
#Sta/Elev= 30
  3969.0  391.09  3980.8  390.58  4097.6  384.28  4399.5  362.62  4458.8  360.50
  4800.8  361.29  4821.6  359.46  4829.5  353.19  4835.9  353.35  4843.9  360.92
  4850.3  361.62  4899.9  360.92  4957.4  362.83  4963.8  354.94  4974.9  351.98
  4977.1  351.48  4997.4  351.98  4999.7  355.31  5002.3  355.31  5010.0  360.92
  5041.0  361.60  5257.4  362.34  5430.1  359.87  5924.9  359.92  6010.1  367.55
  6053.7  370.28  6213.5  387.16  6308.8  395.17  6342.3  397.26  6442.8  398.86
#Mann=6,-1,0
  3969.0     0.1       0  3980.8    0.12       0  4399.5     0.1       0
  4974.9    0.07       0  4997.4     0.1       0  6010.1    0.05       0
Bank Sta=4974.9,4997.4
Exp/Cntr=0.3,0.1

Type RM Length L Ch R = 1,56308,530,530,530
BEGIN DESCRIPTION:
Clear Creek 91.0
END DESCRIPTION:
XS GIS Cut Line= 3
      2754275.99      6799511.03      2753626.00      6800661.00
      2753676.00      6801911.04
#Sta/Elev= 30
  3662.6  383.37  3692.2  375.07  3729.7  368.97  3869.3  367.23  3897.2  365.61
  3984.0  365.85  4037.2  363.72  4226.3  360.82  4429.6  359.90  4722.5  359.76
  4727.3  358.59  4733.1  360.72  4742.3  360.96  4808.2  359.41  4932.3  361.13
  5077.6  359.39  5082.5  359.36  5093.5  360.95  5103.7  360.59  5113.7  356.93
  5122.4  350.82  5124.7  350.32  5144.9  350.82  5153.7  360.78  5376.9  359.53
  5504.0  358.41  5714.1  361.42  5938.5  377.21  6084.4  388.46  6234.6  394.68
#Mann=11,-1,0
  3662.6     0.1       0  3984.0    0.05       0  4429.6    0.12       0
  4722.5     0.1       0  5077.6    0.12       0  5082.5     0.1       0
  5093.5    0.12       0  5122.4    0.07       0  5144.9    0.12       0
  5376.9     0.1       0  5938.5    0.12       0
Bank Sta=5122.4,5144.9
Exp/Cntr=0.3,0.1

Type RM Length L Ch R = 1,55778,1542,1542,1542
BEGIN DESCRIPTION:
Clear Creek 90.0
END DESCRIPTION:
XS GIS Cut Line= 3
      2754176.02      6799410.97      2753226.00      6800861.00
      2753026.01      6801560.97
#Sta/Elev= 30
  3270.3  390.59  3314.1  382.55  3335.1  382.76  3458.8  369.48  3513.7  366.43
  3609.5  363.65  3950.2  359.46  4369.8  359.12  4418.0  358.40  4426.5  356.50
  4462.7  359.43  4822.1  359.53  4828.1  359.38  4960.1  359.41  4969.9  349.91
  4972.2  349.41  4992.4  349.91  4996.3  350.68  5000.8  355.91  5025.9  356.02
  5034.6  358.09  5054.5  359.03  5066.2  355.18  5093.5  352.94  5098.7  353.54
  5107.8  359.12  5171.5  356.67  5187.2  357.60  5232.6  358.72  5731.8  395.59
#Mann=9,-1,0
  3270.3     0.1       0  3513.7    0.05       0  4369.8     0.1       0
  4822.1    0.12       0  4828.1     0.1       0  4969.9    0.07       0
  4992.4     0.1       0  5034.6    0.12       0  5187.2    0.05       0
Bank Sta=4969.9,4992.4
Exp/Cntr=0.3,0.1

Type RM Length L Ch R = 1,54236,1108,1108,1108
BEGIN DESCRIPTION:
Clear Creek 89.0
END DESCRIPTION:
XS GIS Cut Line= 3
      2753876.03      6798760.97      2752626.00      6800061.00
      2752526.00      6801610.97
#Sta/Elev= 30
  3188.6  405.94  3245.1  403.33  3393.8  387.88  3429.1  387.19  3464.6  383.25
  3499.8  383.64  3556.4  378.00  3605.8  375.95  3683.8  367.20  3874.7  359.27
  4106.9  357.08  4468.7  356.60  4518.4  354.52  4673.5  355.93  4730.8  356.12
  4942.6  357.73  4956.7  352.68  4963.9  346.95  4973.6  346.90  4975.9  346.40
  4996.4  346.90  5002.1  356.70  5463.1  356.28  5497.6  360.43  5633.4  370.21
  5803.8  373.62  5984.2  368.40  6054.3  370.03  6401.2  387.62  6545.3  393.53
#Mann=8,-1,0
  3188.6    0.05       0  4106.9    0.12       0  4673.5     0.1       0
  4730.8    0.12       0  4973.6    0.07       0  4996.4    0.12       0
  5497.6    0.05       0  6401.2    0.12       0
Bank Sta=4973.6,4996.4
Exp/Cntr=0.3,0.1

Type RM Length L Ch R = 1,53128,1134,1134,1134
BEGIN DESCRIPTION:
Clear Creek 88.0
END DESCRIPTION:
XS GIS Cut Line= 3
      2753276.03      6798110.96      2752176.00      6799411.00
      2752376.00      6801611.04
#Sta/Elev= 30
  3297.6  398.70  3830.0  367.25  3950.8  362.58  4680.4  354.56  4901.1  354.19
  4922.0  349.01  4929.7  353.60  4944.0  354.94  4997.1  353.98  5019.8  349.36
  5029.0  345.29  5031.3  344.79  5052.5  345.29  5070.9  356.47  5221.5  354.27
  5331.9  354.38  5382.2  356.94  5442.4  354.40  5532.8  356.22  5633.2  354.62
  6133.7  359.08  6285.9  361.76  6326.0  366.45  6366.2  360.13  6446.5  360.15
  6466.6  363.21  6717.6  372.17  6908.4  387.26  7082.2  395.96  7209.7  397.06
#Mann=8,-1,0
  3297.6    0.05       0  4680.4    0.12       0  4997.1     0.1       0
  5019.8    0.12       0  5029.0    0.07       0  5052.5    0.12       0
  6133.7    0.05       0  7082.2    0.12       0
Bank Sta=5029,5052.5
Exp/Cntr=0.3,0.1

Type RM Length L Ch R = 1,51994,1030,1030,1030
BEGIN DESCRIPTION:
Clear Creek 87.0
END DESCRIPTION:
XS GIS Cut Line= 3
      2752926.01      6798210.99      2751376.00      6799511.00
      2750726.03      6800160.97
#Sta/Elev= 30
  2972.9  382.40  3072.4  378.01  3179.1  366.75  3220.9  364.27  3413.3  361.39
  4173.0  354.75  4541.2  354.18  4811.8  352.10  4878.2  352.86  4960.1  354.40
  4967.9  352.37  4974.4  343.67  4977.0  343.20  4979.3  342.70  5000.6  343.20
  5010.0  352.68  5052.5  351.82  5127.6  352.77  5159.1  352.43  5414.3  353.07
  5429.6  354.35  5462.6  354.79  5476.7  352.65  5490.9  343.39  5505.0  351.19
  5519.2  354.76  5557.7  356.10  5660.6  360.87  5816.2  372.24  5915.1  376.99
#Mann=9,-1,0
  2972.9    0.05       0  4878.2     0.1       0  4977.0    0.07       0
  5000.6     0.1       0  5127.6    0.12       0  5159.1    0.05       0
  5414.3     0.1       0  5429.6    0.05       0  5557.7    0.12       0
Bank Sta=4977,5000.6
Exp/Cntr=0.3,0.1

Type RM Length L Ch R = 1,50964,543,543,543
BEGIN DESCRIPTION:
Clear Creek 86.0
END DESCRIPTION:
XS GIS Cut Line= 3
      2753025.97      6798061.02      2750626.00      6799461.00
      2750425.98      6799811.03
#Sta/Elev= 30
  2231.7  388.22  2625.3  365.57  3224.1  359.05  3255.0  359.13  3276.5  352.17
  3292.2  359.60  3537.9  357.38  3563.0  349.42  3575.8  357.27  3615.9  357.43
  3654.0  356.97  3745.4  355.87  4338.7  352.27  4360.6  348.09  4394.5  351.38
  4494.7  351.00  4585.5  346.29  4607.0  351.12  4758.9  351.62  4792.5  351.94
  4932.1  351.58  4952.3  352.12  4974.5  341.77  4977.0  341.27  4999.5  341.77
  5033.2  352.01  5126.1  352.06  5203.2  361.06  5286.5  369.97  5413.3  377.01
#Mann=15,-1,0
  2231.7    0.05       0  3224.1     0.1       0  3537.9    0.12       0
  3615.9    0.05       0  3654.0    0.12       0  3745.4    0.05       0
  4394.5     0.1       0  4494.7    0.05       0  4758.9    0.12       0
  4792.5     0.1       0  4932.1    0.12       0  4974.5    0.07       0
  4999.5    0.12       0  5203.2     0.1       0  5286.5    0.05       0
Bank Sta=4974.5,4999.5
Exp/Cntr=0.3,0.1

Type RM Length L Ch R = 1,50421,578,578,578
BEGIN DESCRIPTION:
Clear Creek 85.0
END DESCRIPTION:
XS GIS Cut Line= 3
      2751726.00      6797511.00      2750476.00      6799111.00
      2750325.99      6799711.03
#Sta/Elev= 30
  2974.2  399.60  3416.5  364.15  3777.0  351.83  3928.8  351.34  4107.0  351.50
  4185.2  352.63  4199.7  346.34  4214.1  352.39  4281.3  351.30  4484.3  348.63
  4535.1  353.74  4550.6  350.76  4556.0  347.81  4607.6  346.88  4641.0  353.34
  4838.4  349.55  4868.9  345.92  4897.9  351.17  4941.1  351.94  4954.0  350.28
  4964.1  341.41  4966.6  340.91  4989.1  341.41  4991.0  347.15  5001.4  351.48
  5027.7  351.18  5243.8  351.04  5354.5  351.68  5489.1  368.58  5623.1  376.72
#Mann=13,-1,0
  2974.2    0.05       0  3777.0    0.12       0  3928.8    0.05       0
  4107.0    0.12       0  4281.3    0.05       0  4550.6     0.1       0
  4607.6    0.05       0  4838.4     0.1       0  4964.1    0.07       0
  4989.1     0.1       0  5027.7    0.05       0  5243.8    0.12       0
  5354.5    0.05       0
Bank Sta=4964.1,4989.1
Exp/Cntr=0.3,0.1

Type RM Length L Ch R = 1,49843,500,500,500
BEGIN DESCRIPTION:
Clear Creek 84.0
END DESCRIPTION:
XS GIS Cut Line= 3
      2751426.01      6797360.98      2750026.00      6798961.00
      2750176.00      6799560.98
#Sta/Elev= 30
  2873.5  397.63  2895.4  395.49  3013.7  386.51  3171.1  377.47  3228.0  371.66
  3397.9  365.08  3596.3  352.23  3963.0  348.44  4170.2  350.06  4184.7  350.45
  4191.4  343.42  4199.0  343.36  4213.2  349.99  4219.8  350.48  4354.6  347.00
  4399.0  348.82  4985.8  350.62  4992.4  349.38  4996.2  346.16  4997.4  341.61
  4999.9  341.11  5022.4  341.61  5040.8  342.30  5051.1  348.92  5058.8  350.85
  5064.0  344.72  5082.0  350.54  5360.3  350.30  5553.6  368.30  5618.0  371.77
#Mann=8,-1,0
  2873.5    0.05       0  2895.4    0.12       0  3013.7    0.05       0
  3963.0    0.12       0  4170.2     0.1       0  4399.0    0.05       0
  4997.4    0.04       0  5022.4    0.05       0
Bank Sta=4997.4,5022.4
Exp/Cntr=0.3,0.1

Type RM Length L Ch R = 1,49343,564,564,564
BEGIN DESCRIPTION:
Clear Creek 83.0
END DESCRIPTION:
XS GIS Cut Line= 3
      2751175.98      6796961.02      2749776.00      6798561.00
      2749375.99      6799661.03
#Sta/Elev= 30
  2866.2  416.93  2930.2  410.78  3071.7  391.01  3178.0  378.14  3369.7  362.04
  3390.6  358.85  3603.2  346.25  4350.3  347.58  4467.8  347.92  4474.5  346.86
  4482.1  341.15  4488.7  342.74  4496.3  347.95  4510.5  345.68  4579.1  346.83
  4962.3  349.17  4978.4  349.54  4985.1  345.24  4989.7  340.00  4992.2  339.50
  5014.7  340.00  5016.5  341.01  5038.1  350.16  5407.2  347.13  5641.3  348.54
  5679.2  350.66  5726.4  349.87  5852.1  355.36  6030.3  370.17  6162.7  375.45
#Mann=7,-1,0
  2866.2    0.05       0  4350.3    0.12       0  4579.1    0.05       0
  4962.3     0.1       0  4989.7    0.07       0  5014.7     0.1       0
  5016.5    0.05       0
Bank Sta=4989.7,5014.7
Exp/Cntr=0.3,0.1

Type RM Length L Ch R = 1,48779,606,606,606
BEGIN DESCRIPTION:
Clear Creek 82.0
END DESCRIPTION:
XS GIS Cut Line= 3
      2751125.99      6796961.01      2749726.00      6798111.00
      2748575.99      6799661.02
#Sta/Elev= 30
  3193.2  410.34  3299.4  396.93  3413.2  379.45  3626.6  357.16  3783.0  346.47
  3875.6  344.43  4720.2  347.10  4731.9  348.05  4777.5  348.16  4791.8  343.12
  4798.3  344.21  4806.2  348.26  4927.3  347.32  4983.4  349.00  4991.3  346.15
  4999.8  340.20  5002.3  339.70  5024.8  340.20  5026.9  346.62  5033.1  348.34
  5136.9  347.09  5905.3  345.84  6226.6  348.15  6291.3  351.39  6426.9  365.07
  6456.1  366.25  6541.7  364.60  6765.0  375.58  6923.3  381.90  6935.0  382.23
#Mann=8,-1,0
  3193.2    0.05       0  4720.2     0.1       0  4731.9    0.12       0
  4999.8    0.07       0  5024.8    0.12       0  5136.9    0.05       0
  6765.0    0.12       0  6923.3    0.05       0
Bank Sta=4999.8,5024.8
Exp/Cntr=0.3,0.1

Type RM Length L Ch R = 1,48173,461,461,461
BEGIN DESCRIPTION:
Clear2
END DESCRIPTION:
XS GIS Cut Line= 3
      2750979.14      6796613.72      2749587.43      6797585.75
      2747175.96      6799061.02
#Sta/Elev= 30
  3288.7  398.57  3605.3  364.59  3919.8  345.77  3999.9  344.63  4910.6  346.02
  4969.5  347.24  4987.5  339.70  4990.0  339.20  5012.5  339.70  5021.2  346.86
  5027.0  343.64  5034.8  347.76  5266.9  345.68  6060.2  348.04  6075.6  343.64
  6081.5  348.10  6102.8  343.29  6133.7  347.89  6139.6  343.87  6155.0  348.41
  6207.1  348.90  7027.7  349.44  7145.0  356.73  7310.1  380.98  7362.3  385.05
  7594.5  384.41  7747.4  391.55  7754.5  392.69  7762.8  400.02  7813.2  399.18
#Mann=7,-1,0
  3288.7    0.05       0  3919.8    0.12       0  3999.9    0.05       0
  4910.6    0.12       0  4987.5    0.07       0  5012.5    0.12       0
  5266.9    0.05       0
Bank Sta=4987.5,5012.5
Exp/Cntr=0.3,0.1

Type RM Length L Ch R = 1,47712,524,524,524
BEGIN DESCRIPTION:
Clear Creek 80.0
END DESCRIPTION:
XS GIS Cut Line= 3
      2750903.24      6796101.00      2749376.00      6797211.00
      2746857.44      6798869.87
#Sta/Elev= 30
  3111.7  401.26  3417.3  373.36  3431.1  368.96  3540.1  377.38  3697.0  377.72
  4010.8  355.56  4663.9  345.19  4992.4  346.08  4994.7  338.67  4997.2  338.17
  5019.7  338.67  5043.4  345.22  5079.5  345.81  6010.1  343.04  6855.7  346.51
  6934.7  347.55  6940.7  352.09  6955.8  353.58  7043.1  349.41  7049.1  352.33
  7115.4  352.07  7202.8  357.48  7208.8  361.07  7244.9  359.38  7425.6  370.73
  7640.2  392.02  7667.2  394.24  7931.6  408.82  7979.9  406.78  8015.5  412.81
#Mann=6,-1,0
  3111.7    0.05       0  4994.7    0.05       0  5019.7    0.05       0
  7640.2   0.075       0  7667.2    0.05       0  7979.9   0.075       0
Bank Sta=4994.7,5019.7
Exp/Cntr=0.3,0.1

Type RM Length L Ch R = 1,47188,555,555,555
BEGIN DESCRIPTION:
Clear Creek 79.0
END DESCRIPTION:
XS GIS Cut Line= 3
      2749226.00      6796360.96      2749176.00      6796761.00
      2746789.94      6798659.59
#Sta/Elev= 30
  4596.9  374.77  4647.3  371.43  4899.3  350.02  4969.8  345.22  4990.0  345.53
  4997.5  339.00  5001.1  338.45  5003.6  337.95  5026.1  338.45  5028.1  344.29
  5036.1  345.57  5050.5  345.92  5164.2  344.38  5362.8  343.69  5668.8  345.22
  5875.4  342.39  6586.6  342.75  6743.5  344.73  7206.4  343.45  7320.2  347.21
  7363.4  350.22  7384.2  352.22  7390.6  353.84  7462.7  358.58  7582.8  372.93
  7725.4  385.85  7911.2  400.13  7996.1  409.25  8010.5  409.86  8049.3  414.84
#Mann=3,-1,0
  4596.9    0.05       0  5001.1    0.04       0  5026.1    0.05       0
Bank Sta=5001.1,5026.1
Exp/Cntr=0.3,0.1

Type RM Length L Ch R = 1,46633,587,587,587
BEGIN DESCRIPTION:
Clear Creek 78.0
END DESCRIPTION:
XS GIS Cut Line= 3
      2749175.95      6796311.01      2748776.00      6796411.00
      2746616.71      6798516.84
#Sta/Elev= 30
  4588.0  377.05  4660.1  368.57  4752.9  359.79  4783.8  354.38  4866.3  349.61
  4907.5  345.14  4948.7  343.11  4977.1  344.01  4982.2  342.61  5000.3  342.87
  5001.8  337.65  5004.3  337.15  5026.8  337.65  5035.6  339.99  5042.6  344.46
  5056.8  345.29  5162.9  343.27  5735.7  341.55  5764.0  342.43  5976.2  341.29
  6948.6  342.20  6967.7  342.20  7085.5  341.58  7171.2  341.95  7250.7  345.78
  7359.4  354.07  7459.5  362.37  7821.8  395.62  7956.2  411.39  8016.4  411.62
#Mann=9,-1,0
  4588.0    0.05       0  5001.8    0.04       0  5026.8    0.05       0
  6948.6    0.12       0  6967.7    0.05       0  7085.5    0.12       0
  7250.7    0.05       0  7359.4    0.12       0  7459.5    0.05       0
Bank Sta=5001.8,5026.8
Exp/Cntr=0.3,0.1

Type RM Length L Ch R = 1,46046,557,557,557
BEGIN DESCRIPTION:
Clear Creek 77.0
END DESCRIPTION:
XS GIS Cut Line= 3
      2749126.00      6795411.00      2748326.00      6796061.00
      2746725.98      6797311.02
#Sta/Elev= 30
  3964.1  391.14  4177.4  374.66  4284.5  364.17  4390.0  358.20  4412.3  355.58
  4717.6  345.25  4732.0  343.45  4888.6  341.89  5008.5  344.19  5016.6  342.10
  5018.5  336.29  5021.0  335.79  5043.5  336.29  5045.5  336.44  5051.9  342.83
  5058.3  341.54  5072.7  343.97  5116.1  341.91  5308.7  343.04  5372.9  341.73
  5393.7  342.98  6234.8  340.43  6270.1  341.82  6384.0  351.90  6462.7  361.42
  6562.2  366.13  6647.2  373.37  6690.6  374.28  6790.1  381.08  7025.3  389.06
#Mann=3,-1,0
  3964.1    0.05       0  5018.5    0.04       0  5043.5    0.05       0
Bank Sta=5018.5,5043.5
Exp/Cntr=0.3,0.1

Type RM Length L Ch R = 1,45489,598,598,598
BEGIN DESCRIPTION:
Clear Creek 76.0
END DESCRIPTION:
XS GIS Cut Line= 3
      2748476.01      6794960.99      2747876.00      6795761.00
      2746576.01      6797310.99
#Sta/Elev= 30
  4007.8  380.65  4035.9  378.82  4285.9  355.73  4435.9  344.54  4494.6  342.79
  4550.5  341.55  4690.7  341.96  4771.4  341.65  4929.7  343.46  4935.9  342.54
  4944.3  343.10  4950.5  341.55  4957.8  342.80  4965.1  339.48  4967.2  335.99
  4969.7  335.49  4992.2  335.99  4994.3  339.37  5000.5  341.13  5021.5  343.18
  5113.9  341.28  5569.0  340.01  6292.5  343.21  6405.7  349.51  6413.5  351.18
  6526.7  362.42  6576.1  370.63  6668.5  381.49  6988.5  392.42  7030.8  391.53
#Mann=5,-1,0
  4007.8    0.05       0  4494.6    0.12       0  4690.7    0.05       0
  4967.2    0.05       0  4992.2    0.05       0
Bank Sta=4967.2,4992.2
Exp/Cntr=0.3,0.1

Type RM Length L Ch R = 1,44891,489,489,489
BEGIN DESCRIPTION:
Clear Creek 75.0
END DESCRIPTION:
XS GIS Cut Line= 3
      2748141.13      6794734.05      2747574.44      6795316.87
      2746126.01      6795711.00
#Sta/Elev= 30
  4187.1  352.10  4246.4  350.84  4365.6  347.41  4485.6  343.36  4616.0  345.02
  4754.4  351.68  4775.5  348.86  4888.7  345.72  4952.3  339.86  4973.6  340.13
  4987.0  343.64  4994.7  340.23  4996.2  335.26  4998.7  334.76  5021.2  335.26
  5034.7  342.68  5181.4  341.18  5231.7  340.58  5361.1  340.63  5540.0  343.66
  5558.0  341.21  5565.6  335.99  5570.8  335.66  5578.7  336.42  5589.1  342.97
  5674.9  342.99  5698.0  342.79  6215.8  340.92  6369.7  353.75  6501.1  371.99
#Mann=13,-1,0
  4187.1    0.12       0  4246.4    0.05       0  4365.6    0.12       0
  4616.0    0.05       0  4987.0     0.1       0  4996.2    0.07       0
  5021.2     0.1       0  5181.4    0.12       0  5231.7     0.1       0
  5361.1    0.12       0  5540.0    0.05       0  5674.9    0.12       0
  5698.0    0.05       0
Bank Sta=4996.2,5021.2
Exp/Cntr=0.3,0.1

Type RM Length L Ch R = 1,44402,561,561,561
BEGIN DESCRIPTION:
Clear Creek 74.0
END DESCRIPTION:
XS GIS Cut Line= 3
      2748478.70      6794335.52      2747226.00      6795011.00
      2745776.00      6795511.00
#Sta/Elev= 30
  3576.8  370.18  3645.7  360.45  3871.2  353.38  3898.8  350.08  4002.6  352.12
  4096.8  349.48  4166.4  344.17  4232.1  347.18  4483.4  341.17  4750.1  339.23
  4991.9  342.37  4997.2  338.81  4997.8  334.84  5000.3  334.34  5022.8  334.84
  5046.8  342.00  5211.6  339.25  5309.8  341.57  5338.5  340.27  5348.3  336.15
  5353.6  341.72  5359.7  336.67  5370.2  336.68  5379.5  342.02  5416.0  342.79
  5868.6  339.90  5917.6  339.61  6060.7  341.67  6393.4  374.23  6533.8  380.28
#Mann=8,-1,0
  3576.8    0.05       0  3645.7    0.12       0  4096.8    0.05       0
  4997.8    0.04       0  5022.8    0.05       0  5309.8    0.05       0
  5868.6    0.12       0  5917.6    0.05       0
Bank Sta=4997.8,5022.8
Exp/Cntr=0.3,0.1

Type RM Length L Ch R = 1,43841,566,566,566
BEGIN DESCRIPTION:
Clear Creek 73.0
END DESCRIPTION:
XS GIS Cut Line= 3
      2748704.17      6794015.35      2746826.00      6794661.00
      2745577.44      6795076.41
#Sta/Elev= 30
  3009.6  377.46  3073.0  375.45  3137.2  374.99  3163.2  370.40  3178.5  371.85
  3199.7  370.11  3231.0  374.48  3288.2  367.01  3444.4  359.61  3494.1  355.32
  3515.2  355.76  3532.8  352.04  3538.1  354.50  3569.3  353.80  3595.3  349.90
  3814.0  348.00  4084.6  341.85  4423.0  339.24  4998.3  342.08  5006.2  341.09
  5014.8  334.16  5017.3  333.66  5039.8  334.16  5048.4  341.60  5058.9  341.87
  5618.0  338.68  5966.1  358.86  6087.4  371.26  6219.3  372.84  6311.5  381.53
#Mann=5,-1,0
  3009.6    0.05       0  3073.0    0.12       0  3178.5    0.05       0
  5014.8    0.04       0  5039.8    0.05       0
Bank Sta=5014.8,5039.8
Exp/Cntr=0.3,0.1
