HEC-RAS study Clear Creek.prj: Clear Creek Base Level Engineering

--- Clear Creek.g01 (geometry) --- (continued)

Type RM Length L Ch R = 1,43275,520,520,520
BEGIN DESCRIPTION:
Clear Creek 72.0
END DESCRIPTION:
XS GIS Cut Line= 3
      2748527.87      6793269.89      2746576.00      6794211.00
      2745776.01      6794711.00
#Sta/Elev= 30
  2833.2  385.01  2857.5  383.60  2872.2  381.25  2879.7  377.25  2885.1  377.96
  2904.4  378.30  2934.5  377.59  2979.6  370.62  3007.9  367.89  3217.0  351.13
  3330.0  343.85  3397.9  341.92  3778.9  337.23  4012.1  336.73  4183.4  337.33
  4279.4  339.76  4799.6  337.59  4977.9  340.51  4986.0  335.78  4991.6  338.85
  4997.3  334.35  5016.5  333.64  5019.0  333.14  5041.5  333.64  5044.3  340.73
  5206.3  338.02  5254.0  338.43  5579.7  342.40  5747.2  355.76  5943.5  378.65
#Mann=7,-1,0
  2833.2    0.05       0  2885.1    0.12       0  2904.4    0.05       0
  5016.5    0.04       0  5041.5    0.05       0  5206.3     0.1       0
  5254.0    0.05       0
Bank Sta=5016.5,5041.5
Exp/Cntr=0.3,0.1

Type RM Length L Ch R = 1,42755,575,575,575
BEGIN DESCRIPTION:
Clear Creek 71.0
END DESCRIPTION:
XS GIS Cut Line= 3
      2748026.04      6792610.97      2746476.00      6793761.00
      2745675.98      6794111.01
#Sta/Elev= 30
  3060.9  387.24  3147.6  378.60  3174.6  373.55  3197.6  370.91  3203.9  369.06
  3224.7  367.68  3247.7  364.54  3260.2  360.87  3283.2  359.54  3324.9  352.75
  3333.3  352.82  3418.8  344.25  3468.9  341.98  3804.8  334.00  4076.0  335.57
  4754.4  336.67  5005.4  339.76  5016.3  333.07  5018.8  332.57  5041.3  333.07
  5045.5  339.50  5122.0  339.14  5174.6  337.46  5378.1  340.71  5448.2  344.13
  5523.9  344.44  5599.5  346.96  5698.5  353.51  5756.2  360.22  5864.2  365.56
#Mann=3,-1,0
  3060.9    0.05       0  5016.3    0.04       0  5041.3    0.05       0
Bank Sta=5016.3,5041.3
Exp/Cntr=0.3,0.1

Type RM Length L Ch R = 1,42180,544,544,544
BEGIN DESCRIPTION:
Clear Creek 70.0
END DESCRIPTION:
XS GIS Cut Line= 3
      2747925.97      6792561.01      2746376.00      6793261.00
      2745576.01      6793610.99
#Sta/Elev= 30
  3299.2  381.47  3336.6  378.69  3397.9  371.49  3406.0  369.11  3452.2  362.81
  3480.8  356.58  3486.3  356.86  3509.4  352.92  3540.6  352.41  3639.3  343.35
  3844.1  337.71  3919.8  333.98  4010.6  333.98  4780.5  335.89  4991.1  338.54
  5002.6  338.03  5008.9  334.36  5009.2  332.51  5011.7  332.01  5034.2  332.51
  5037.7  337.39  5043.6  338.55  5264.6  336.36  5462.6  336.87  5637.3  350.86
  5660.7  354.42  5736.3  361.02  5783.1  368.09  5835.3  374.11  5873.1  377.12
#Mann=5,-1,0
  3299.2    0.05       0  3919.8    0.12       0  4010.6    0.05       0
  5009.2    0.04       0  5034.2    0.05       0
Bank Sta=5009.2,5034.2
Exp/Cntr=0.3,0.1

Type RM Length L Ch R = 1,41636,561,561,561
BEGIN DESCRIPTION:
Clear Creek 69.0
END DESCRIPTION:
XS GIS Cut Line= 3
      2747275.98      6791511.02      2746326.00      6792811.00
      2745576.01      6793510.99
#Sta/Elev= 30
  3385.4  390.33  3388.5  390.33  3392.7  385.66  3413.6  380.95  3528.6  369.89
  3664.5  363.10  3771.1  360.04  3850.6  354.69  3871.5  355.50  3900.8  351.80
  3915.5  351.45  3921.7  353.31  3951.0  348.52  4036.8  342.41  4151.8  336.71
  4207.7  335.63  4333.0  334.10  4388.1  333.21  4415.2  334.62  4946.0  337.52
  5016.7  333.19  5032.6  330.70  5035.1  330.20  5057.6  330.70  5066.1  337.63
  5214.6  334.89  5618.1  335.49  5646.5  336.86  5851.6  361.58  6021.4  378.04
#Mann=5,-1,0
  3385.4    0.05       0  4207.7    0.12       0  4333.0    0.05       0
  5032.6    0.05       0  5057.6    0.05       0
Bank Sta=5032.6,5057.6
Exp/Cntr=0.3,0.1

Type RM Length L Ch R = 1,41075,545,545,545
BEGIN DESCRIPTION:
Clear Creek 68.0
END DESCRIPTION:
XS GIS Cut Line= 3
      2746926.02      6791710.98      2746126.00      6792411.00
      2745426.00      6793661.00
#Sta/Elev= 30
  3941.1  370.70  3976.7  369.70  4040.3  364.29  4232.0  353.16  4252.9  350.29
  4342.2  344.06  4500.6  334.79  4632.0  334.93  4643.0  334.93  4649.7  332.84
  4655.4  334.50  4776.5  334.34  4833.8  333.77  4947.7  336.85  4961.9  336.37
  4968.6  333.16  4970.3  330.64  4972.8  330.14  4995.3  330.64  4997.0  333.64
  5000.8  336.71  5038.8  336.20  5051.6  336.02  5267.8  334.28  5834.1  334.65
  5915.1  341.82  6127.3  369.12  6217.6  376.83  6342.0  380.49  6436.8  380.10
#Mann=9,-1,0
  3941.1    0.05       0  4342.2    0.12       0  4632.0     0.1       0
  4655.4    0.12       0  4776.5    0.05       0  4970.3    0.04       0
  4995.3    0.05       0  5038.8    0.12       0  5051.6    0.05       0
Bank Sta=4970.3,4995.3
Exp/Cntr=0.3,0.1

Type RM Length L Ch R = 1,40530,509,509,509
BEGIN DESCRIPTION:
Clear Creek 67.0
END DESCRIPTION:
XS GIS Cut Line= 3
      2746937.82      6791451.13      2746226.00      6791961.00
      2744626.03      6793060.98
#Sta/Elev= 30
  4129.2  373.14  4294.8  372.76  4538.0  361.72  4905.6  334.14  4976.5  335.49
  4982.7  333.65  4984.9  330.31  4987.4  329.81  5009.9  330.31  5018.3  336.45
  5095.1  335.49  5346.8  334.95  5508.1  333.94  5537.9  337.50  5544.0  334.80
  5573.8  333.40  5623.7  333.62  5636.7  333.97  5645.5  338.07  5672.5  339.22
  5681.3  336.05  5708.6  333.94  6147.4  335.65  6314.6  346.67  6356.5  347.19
  6514.8  359.21  6601.4  368.96  6643.3  367.75  6846.3  378.30  6946.4  378.52
#Mann=6,-1,0
  4129.2    0.05       0  4905.6     0.1       0  4984.9    0.07       0
  5009.9     0.1       0  5095.1    0.12       0  5346.8    0.05       0
Bank Sta=4984.9,5009.9
Exp/Cntr=0.3,0.1

Type RM Length L Ch R = 1,40021,543,543,543
BEGIN DESCRIPTION:
Clear Creek 66.0
END DESCRIPTION:
XS GIS Cut Line= 3
      2746793.31      6790997.67      2745976.00      6791561.00
      2744276.26      6792426.39
#Sta/Elev= 30
  4007.6  375.10  4088.0  369.66  4115.0  364.18  4180.6  363.10  4195.5  366.05
  4222.9  361.40  4374.7  351.07  4490.1  345.43  4539.0  341.02  4819.4  334.10
  4864.3  332.91  4971.8  335.78  4977.9  334.77  4984.7  330.03  4987.2  329.53
  5009.7  330.03  5014.2  336.00  5053.0  334.38  5192.1  335.09  5314.3  331.89
  5387.4  332.63  5492.3  331.94  5809.3  335.57  6308.4  346.03  6404.2  348.39
  6479.2  352.71  6621.0  361.36  6637.6  364.05  6704.3  368.55  6907.6  372.70
#Mann=7,-1,0
  4007.6    0.05       0  4819.4    0.12       0  4984.7    0.07       0
  5009.7    0.12       0  5387.4    0.05       0  6308.4    0.12       0
  6479.2    0.05       0
Bank Sta=4984.7,5009.7
Exp/Cntr=0.3,0.1

Type RM Length L Ch R = 1,39478,549,549,549
BEGIN DESCRIPTION:
Clear Creek 65.0
END DESCRIPTION:
XS GIS Cut Line= 3
      2746526.05      6790860.99      2745726.00      6791111.00
      2744426.00      6791311.00
#Sta/Elev= 30
  4165.9  376.67  4247.1  367.09  4447.3  348.64  4626.9  337.32  4670.8  336.35
  4690.3  337.78  4722.8  332.01  4805.0  333.42  4836.5  335.68  4846.9  335.16
  4852.7  333.19  4880.3  332.15  4987.9  335.47  4993.6  334.83  5001.5  329.67
  5011.8  328.90  5014.3  328.40  5036.8  328.90  5038.2  334.98  5400.0  331.65
  5621.3  333.18  5773.0  336.16  5854.0  335.47  5965.3  338.80  6090.5  345.87
  6158.8  352.01  6217.0  359.69  6268.8  364.44  6285.2  367.37  6319.4  369.95
#Mann=6,-1,0
  4165.9    0.05       0  4670.8     0.1       0  4880.3    0.12       0
  5011.8    0.07       0  5036.8    0.12       0  5400.0    0.05       0
Bank Sta=5011.8,5036.8
Exp/Cntr=0.3,0.1

Type RM Length L Ch R = 1,38929,1619,1619,1619
BEGIN DESCRIPTION:
Clear Creek 64.0
END DESCRIPTION:
XS GIS Cut Line= 3
      2746568.90      6790727.91      2745526.00      6790661.00
      2744376.03      6791160.99
#Sta/Elev= 30
  3949.5  376.65  4433.4  340.39  4553.6  333.75  4599.2  332.82  4714.0  331.09
  4834.2  331.83  4894.3  334.35  4917.9  332.44  5003.5  332.51  5048.8  327.65
  5051.3  327.15  5073.8  327.65  5079.3  327.77  5102.8  334.17  5108.2  334.43
  5131.7  332.93  5277.8  332.49  5283.2  333.58  5343.5  331.70  5613.8  330.99
  5633.3  331.37  5662.2  334.77  5680.1  334.35  5685.6  332.34  5709.0  334.14
  5746.9  332.25  5784.8  333.94  6035.6  355.30  6187.2  374.54  6248.5  376.63
#Mann=5,-1,0
  3949.5    0.05       0  4599.2    0.12       0  5048.8    0.07       0
  5073.8    0.12       0  5613.8    0.05       0
Bank Sta=5048.8,5073.8
Exp/Cntr=0.3,0.1

Type RM Length L Ch R = 1,37310,550,550,550
BEGIN DESCRIPTION:
Clear Creek 63.0
END DESCRIPTION:
XS GIS Cut Line= 3
      2746505.37      6790242.67      2744826.00      6789861.00
      2744076.04      6790210.98
#Sta/Elev= 30
  3278.1  363.75  3305.6  360.98  3353.8  359.68  3544.1  343.24  3622.5  338.29
  3848.1  331.51  3931.8  331.39  4045.2  331.26  4148.6  330.42  4272.2  331.01
  4436.5  329.77  4553.8  329.16  4643.2  329.36  4867.0  329.48  4969.5  331.38
  4976.2  330.84  4981.3  327.22  5002.0  325.55  5004.5  325.05  5027.0  325.55
  5031.8  331.68  5099.6  330.11  5105.9  331.95  5128.8  332.06  5437.0  329.09
  5585.2  341.79  5630.9  348.22  5648.2  349.44  5750.7  362.70  5827.9  371.26
#Mann=9,-1,0
  3278.1    0.05       0  3931.8    0.12       0  4045.2    0.05       0
  4148.6    0.12       0  4436.5     0.1       0  4553.8    0.12       0
  4643.2     0.1       0  5002.0    0.07       0  5027.0     0.1       0
Bank Sta=5002,5027
Exp/Cntr=0.3,0.1

Type RM Length L Ch R = 1,36760,509,509,509
BEGIN DESCRIPTION:
Clear Creek 62.0
END DESCRIPTION:
XS GIS Cut Line= 3
      2746276.02      6787860.97      2744726.00      6789461.00
      2744075.99      6789611.00
#Sta/Elev= 30
  2776.7  375.61  3215.2  340.99  3377.8  334.24  4650.8  329.57  4721.6  324.73
  4728.5  328.03  4742.7  329.76  4799.3  327.68  4855.9  331.11  4870.0  327.07
  4877.2  328.67  4884.1  324.31  4891.2  325.34  4913.9  323.80  4916.4  323.30
  4939.3  323.80  4947.9  329.07  4954.9  327.68  4962.1  331.39  4990.4  330.79
  4997.3  324.43  5000.9  323.98  5014.7  323.92  5028.3  331.24  5119.0  328.95
  5183.6  330.32  5342.2  328.24  5428.6  330.53  5555.8  344.60  5671.5  359.36
#Mann=7,-1,0
  2776.7    0.05       0  4891.2    0.12       0  4913.9    0.07       0
  4939.3    0.12       0  5183.6     0.1       0  5342.2    0.12       0
  5555.8    0.05       0
Bank Sta=4913.9,4939.3
Exp/Cntr=0.3,0.1

Type RM Length L Ch R = 1,36251,552,552,552
BEGIN DESCRIPTION:
Clear Creek 61.0
END DESCRIPTION:
XS GIS Cut Line= 3
      2746026.02      6787710.98      2744476.00      6789161.00
      2744076.01      6789560.99
#Sta/Elev= 30
  2877.0  362.67  2954.9  354.57  3124.5  344.31  3421.9  333.61  3584.6  331.39
  3726.0  331.41  3733.1  330.15  4190.3  327.77  4235.3  327.38  4277.8  324.78
  4306.1  325.89  4320.3  328.02  4330.1  327.27  4645.6  328.39  4673.9  329.86
  4819.3  328.88  4949.9  330.32  4957.3  327.00  4958.7  322.97  4961.2  322.47
  4984.2  322.97  5003.1  323.61  5013.7  328.77  5101.3  329.05  5163.4  330.09
  5244.6  330.40  5282.4  330.45  5367.2  336.60  5466.2  347.36  5565.2  361.09
#Mann=9,-1,0
  2877.0    0.05       0  4190.3    0.12       0  4330.1    0.05       0
  4819.3    0.12       0  4958.7    0.07       0  4984.2    0.12       0
  5101.3    0.05       0  5163.4    0.12       0  5244.6    0.05       0
Bank Sta=4958.7,4984.2
Exp/Cntr=0.3,0.1

Type RM Length L Ch R = 1,35699,569,569,569
BEGIN DESCRIPTION:
Clear Creek 60.0
END DESCRIPTION:
XS GIS Cut Line= 3
      2745800.76      6786976.86      2744426.00      6788661.00
      2743625.98      6789111.01
#Sta/Elev= 30
  2826.5  376.38  2967.9  367.98  3060.5  366.60  3124.4  360.06  3237.9  356.66
  3479.1  343.80  3792.1  332.51  4006.1  327.73  4339.5  327.18  4432.5  328.13
  4445.5  325.06  4583.8  326.79  4937.6  328.90  4972.5  329.84  4979.0  327.91
  4980.6  322.83  4983.1  322.33  5006.1  322.83  5008.5  327.48  5014.4  329.54
  5148.7  331.08  5170.4  335.29  5197.8  345.86  5300.4  341.83  5375.6  342.29
  5462.3  338.36  5602.5  337.89  5661.8  335.23  5786.1  341.02  5918.4  353.34
#Mann=7,-1,0
  2826.5    0.05       0  4339.5    0.12       0  4583.8    0.05       0
  4937.6    0.12       0  4980.6    0.07       0  5006.1    0.12       0
  5014.4    0.05       0
Bank Sta=4980.6,5006.1
Exp/Cntr=0.3,0.1

Type RM Length L Ch R = 1,35130,556,556,556
BEGIN DESCRIPTION:
Clear Creek 59.0
END DESCRIPTION:
XS GIS Cut Line= 3
      2745376.03      6786810.97      2744126.00      6788261.00
      2743476.02      6789060.97
#Sta/Elev= 30
  3081.1  398.12  3244.1  392.21  3407.5  379.17  3627.0  370.16  3747.6  358.39
  3882.6  337.22  3989.0  328.69  4144.8  331.16  4194.1  326.18  4300.6  327.03
  4314.8  325.24  4335.7  327.29  4967.6  328.29  4975.7  322.58  4978.2  322.08
  5001.2  322.58  5017.1  322.97  5023.6  327.40  5031.5  324.83  5037.9  328.23
  5045.9  324.60  5052.3  327.99  5066.7  323.22  5081.0  323.48  5087.5  328.61
  5429.4  328.11  5464.6  331.26  5528.5  330.99  5806.6  346.32  6026.3  366.36
#Mann=3,-1,0
  3081.1    0.05       0  4975.7    0.04       0  5001.2    0.05       0
Bank Sta=4975.7,5001.2
Exp/Cntr=0.3,0.1

Type RM Length L Ch R = 1,34574,512,512,512
BEGIN DESCRIPTION:
Clear Creek 58.0
END DESCRIPTION:
XS GIS Cut Line= 3
      2745126.00      6787011.00      2743876.00      6788011.00
      2743125.97      6788511.02
#Sta/Elev= 30
  3387.7  383.81  3451.7  383.06  3551.8  378.02  3657.4  367.80  3735.9  363.95
  3764.7  361.61  3779.1  356.48  3863.9  344.59  3942.4  336.18  4120.1  326.73
  4177.7  327.45  4198.5  325.40  4270.5  324.58  4305.7  324.81  4326.6  327.30
  4398.6  324.89  4779.6  327.09  4921.0  327.23  4981.3  327.94  4983.2  322.62
  4985.8  322.12  5008.7  322.62  5074.1  322.93  5083.1  326.36  5096.6  327.65
  5434.7  325.87  5572.9  330.04  5593.9  332.98  5738.1  344.18  5889.9  361.31
#Mann=5,-1,0
  3387.7    0.05       0  4779.6     0.1       0  4921.0    0.05       0
  4983.2    0.04       0  5008.7    0.05       0
Bank Sta=4983.2,5008.7
Exp/Cntr=0.3,0.1

Type RM Length L Ch R = 1,34062,1067,1067,1067
BEGIN DESCRIPTION:
Clear Creek 57.0
END DESCRIPTION:
XS GIS Cut Line= 3
      2745008.99      6786677.45      2743776.00      6787761.00
      2743075.97      6788511.03
#Sta/Elev= 30
  3358.3  380.20  3519.1  373.09  3568.4  373.87  3632.0  371.70  3731.6  361.60
  3852.1  352.03  3936.6  347.46  4001.1  341.59  4050.4  339.83  4071.3  337.23
  4163.3  331.77  4319.9  325.88  4560.4  325.35  4574.2  323.84  4638.7  325.48
  4917.6  326.22  4971.7  326.84  4986.0  326.63  4992.6  325.13  5003.2  326.40
  5008.2  323.13  5010.8  322.63  5033.7  323.13  5035.2  326.63  5042.0  326.81
  5267.5  326.94  5629.2  325.80  5756.7  335.64  5983.4  362.04  6025.7  365.08
#Mann=5,-1,0
  3358.3    0.05       0  4917.6     0.1       0  5008.2    0.07       0
  5033.7     0.1       0  5267.5    0.05       0
Bank Sta=5008.2,5033.7
Exp/Cntr=0.3,0.1

Type RM Length L Ch R = 1,32995,549,549,549
BEGIN DESCRIPTION:
Clear Creek 56.0
END DESCRIPTION:
XS GIS Cut Line= 3
      2744828.30      6786231.56      2743326.00      6787211.00
      2742926.00      6788611.00
#Sta/Elev= 30
  3206.2  367.99  3229.8  366.36  3250.8  356.30  3256.8  362.18  3266.0  360.23
  3271.9  363.77  3280.6  361.29  3287.1  355.81  3293.0  359.63  3308.2  361.92
  3398.5  355.99  3634.1  344.30  4290.8  324.23  4385.5  322.79  4414.6  326.00
  4626.3  324.89  4992.0  325.46  5002.2  325.23  5003.7  322.71  5006.3  322.21
  5029.2  322.71  5050.3  325.94  5141.5  324.69  5650.9  325.11  5860.6  325.42
  5904.4  325.26  5935.6  329.83  6029.2  333.32  6360.7  365.48  6455.6  366.03
#Mann=9,-1,0
  3206.2    0.12       0  3398.5    0.05       0  4290.8    0.12       0
  4626.3     0.1       0  5003.7    0.07       0  5029.2     0.1       0
  5141.5    0.05       0  5650.9    0.12       0  5860.6    0.05       0
Bank Sta=5003.7,5029.2
Exp/Cntr=0.3,0.1

Type RM Length L Ch R = 1,32446,495,495,495
BEGIN DESCRIPTION:
Clear Creek 55.0
END DESCRIPTION:
XS GIS Cut Line= 3
      2744626.02      6785910.99      2743076.00      6786761.00
      2741776.02      6787560.99
#Sta/Elev= 30
  3236.6  362.16  3320.9  353.84  3401.8  347.44  3516.1  340.15  3644.7  334.49
  4142.1  324.56  4445.5  325.19  4467.0  322.38  4469.6  321.88  4492.5  322.38
  4495.9  325.71  4650.8  323.32  4981.6  324.83  4990.6  322.80  4996.3  324.98
  5001.5  322.72  5048.8  325.15  5427.1  323.09  5857.4  325.62  5937.4  327.16
  5971.7  327.77  5991.8  328.63  6007.2  327.01  6014.2  322.61  6028.5  322.96
  6043.9  328.36  6076.0  327.92  6159.9  327.82  6306.6  337.33  6530.8  361.68
#Mann=12,-1,0
  3236.6    0.05       0  3320.9    0.12       0  3401.8     0.1       0
  3516.1    0.12       0  3644.7    0.05       0  4142.1     0.1       0
  4467.0    0.07       0  4492.5     0.1       0  5857.4    0.12       0
  5937.4     0.1       0  5971.7    0.12       0  6076.0    0.05       0
Bank Sta=4467,4492.5
Exp/Cntr=0.3,0.1

Type RM Length L Ch R = 1,31951,590,590,590
BEGIN DESCRIPTION:
Clear Creek 54.0
END DESCRIPTION:
XS GIS Cut Line= 3
      2744226.00      6785011.00      2742826.00      6786461.00
      2741676.04      6787560.97
#Sta/Elev= 30
  2963.8  364.64  2991.0  362.09  3033.5  356.75  3140.7  342.84  3289.0  328.83
  3338.7  324.34  3432.8  322.62  3502.7  321.85  3505.3  321.35  3528.2  321.85
  3565.8  322.29  3721.3  322.36  4165.3  322.61  4838.0  322.33  4922.9  324.46
  4951.2  322.27  5085.5  324.57  5311.6  321.95  5799.7  327.49  5807.0  323.09
  5813.9  322.77  5835.3  325.86  5842.2  323.38  5849.4  327.57  5874.5  327.22
  6040.3  326.31  6202.9  333.01  6294.8  341.39  6450.5  359.99  6570.7  369.72
#Mann=11,-1,0
  2963.8    0.05       0  2991.0     0.1       0  3033.5    0.12       0
  3289.0    0.05       0  3432.8    0.12       0  3502.7    0.07       0
  3528.2    0.12       0  3565.8     0.1       0  3721.3    0.12       0
  4165.3     0.1       0  5874.5    0.05       0
Bank Sta=3502.7,3528.2
Exp/Cntr=0.3,0.1

Type RM Length L Ch R = 1,31361,509,509,509
BEGIN DESCRIPTION:
Clear Creek 53.0
END DESCRIPTION:
XS GIS Cut Line= 3
      2743976.02      6784860.99      2742576.00      6786011.00
      2741425.97      6787411.03
#Sta/Elev= 30
  3184.7  365.18  3255.8  355.76  3334.0  349.47  3483.8  332.38  3539.9  327.36
  3618.1  325.25  4023.3  323.92  4574.8  322.39  4669.7  322.16  4713.2  321.73
  4715.7  321.23  4738.8  321.73  4802.9  322.25  4904.6  323.50  5230.3  322.49
  5377.2  322.57  5438.5  323.00  5536.8  324.50  5543.3  322.16  5599.1  324.65
  6019.0  322.73  6140.2  323.43  6275.8  327.46  6346.2  331.60  6467.4  342.69
  6502.6  343.58  6510.5  345.77  6588.3  351.09  6758.0  369.13  6808.3  371.60
#Mann=12,-1,0
  3184.7     0.1       0  3483.8    0.05       0  4023.3    0.12       0
  4574.8    0.05       0  4669.7    0.12       0  4713.2    0.07       0
  4738.8    0.12       0  4802.9     0.1       0  5230.3    0.12       0
  5377.2     0.1       0  5438.5    0.12       0  5599.1    0.05       0
Bank Sta=4713.2,4738.8
Exp/Cntr=0.3,0.1

Type RM Length L Ch R = 1,30852,565,565,565
BEGIN DESCRIPTION:
Clear Creek 52.0
END DESCRIPTION:
XS GIS Cut Line= 3
      2743725.97      6784811.02      2742176.00      6785961.00
      2741078.48      6786626.85
#Sta/Elev= 30
  3070.0  350.26  3106.5  348.26  3112.7  349.85  3127.4  347.65  3133.6  348.95
  3156.6  347.12  3162.8  348.48  3233.7  339.91  3313.0  334.26  3348.5  329.16
  3398.6  326.40  3692.6  325.66  3749.1  324.66  3770.0  322.27  3820.0  322.04
  4574.1  322.10  4807.7  322.50  4823.0  321.86  4825.6  321.36  4849.5  321.86
  4913.4  323.02  4987.6  322.00  5059.2  322.22  5082.1  322.32  5422.6  322.00
  5434.4  322.00  5786.0  322.46  5904.2  328.27  6011.9  335.45  6283.7  361.56
#Mann=12,-1,0
  3070.0    0.05       0  4574.1     0.1       0  4807.7    0.12       0
  4823.0    0.05       0  4849.5    0.12       0  4987.6    0.05       0
  5059.2    0.12       0  5082.1    0.05       0  5422.6    0.12       0
  5434.4    0.05       0  5786.0    0.12       0  5904.2    0.05       0
Bank Sta=4823,4849.5
Exp/Cntr=0.3,0.1

Type RM Length L Ch R = 1,30287,564,564,564
BEGIN DESCRIPTION:
Clear Creek 51.0
END DESCRIPTION:
XS GIS Cut Line= 3
      2743425.98      6783911.02      2741876.00      6785511.00
      2740977.05      6785721.03
#Sta/Elev= 30
  2777.0  354.02  2779.3  354.02  2845.0  348.45  3026.2  334.56  3187.1  332.06
  3208.5  326.65  3222.5  327.03  3229.6  331.30  3260.1  331.18  3286.2  328.46
  3328.6  332.03  3384.9  330.52  3448.8  329.91  3455.9  326.80  3482.3  329.08
  3548.5  329.63  3784.7  327.60  3918.0  325.04  4051.3  324.85  4201.8  324.89
  4411.3  321.82  4414.0  321.32  4438.1  321.82  4538.6  322.23  5266.2  322.00
  5368.4  322.00  5675.0  338.67  5726.5  341.50  5777.2  344.76  5927.8  358.00
#Mann=20,-1,0
  2777.0     0.1       0  2779.3    0.12       0  2845.0     0.1       0
  3026.2    0.12       0  3260.1     0.1       0  3384.9    0.12       0
  3482.3    0.05       0  3548.5    0.12       0  3784.7     0.1       0
  3918.0    0.12       0  4051.3    0.05       0  4201.8    0.12       0
  4411.3    0.03       0  4438.1    0.12       0  4538.6    0.05       0
  5266.2    0.12       0  5368.4     0.1       0  5675.0    0.12       0
  5726.5     0.1       0  5777.2    0.05       0
Bank Sta=4411.3,4438.1
Exp/Cntr=0.3,0.1

Type RM Length L Ch R = 1,29723,547,547,547
BEGIN DESCRIPTION:
Clear Creek 50.0
END DESCRIPTION:
XS GIS Cut Line= 3
      2743226.00      6783411.00      2741676.00      6785011.00
      2741075.99      6785311.00
#Sta/Elev= 30
  2776.9  369.52  2962.9  356.52  3004.8  353.17  3088.0  347.76  3095.2  348.44
  3170.0  342.42  3259.0  337.92  3315.9  334.81  3406.2  331.28  3427.6  331.64
  3455.9  329.76  3675.0  326.44  4021.5  324.89  4190.7  322.80  4298.0  322.00
  4300.7  321.50  4674.2  321.68  5275.4  321.99  5285.6  322.00  5309.2  322.19
  5317.6  325.48  5326.0  335.93  5331.6  334.57  5388.7  339.73  5488.1  344.51
  5541.2  348.82  5567.2  349.25  5586.0  349.48  5594.3  353.32  5675.4  361.80
#Mann=13,-1,0
  2776.9    0.12       0  2962.9     0.1       0  3004.8    0.12       0
  3170.0    0.05       0  3259.0    0.12       0  3315.9    0.05       0
  4190.7    0.12       0  4298.0    0.05       0  4674.2    0.05       0
  5275.4     0.1       0  5285.6    0.12       0  5388.7    0.12       0
  5567.2    0.05       0
Bank Sta=4298,5285.6
Exp/Cntr=0.3,0.1

Type RM Length L Ch R = 1,29176,540,540,540
BEGIN DESCRIPTION:
Clear Creek 49.0
END DESCRIPTION:
XS GIS Cut Line= 3
      2742325.99      6782911.01      2741526.00      6784511.00
      2740975.64      6785106.07
#Sta/Elev= 30
  3211.4  377.67  3286.9  374.00  3323.2  367.52  3337.2  368.08  3627.9  342.92
  3650.2  338.54  3694.9  338.97  3807.0  332.03  3882.2  328.82  3890.6  326.39
  3896.2  328.03  3913.0  322.24  3985.6  322.00  3994.0  324.50  4020.3  324.08
  4098.2  322.00  4385.8  321.56  4422.3  321.50  4456.3  321.50  5306.0  321.96
  5376.9  322.00  5389.5  322.00  5424.6  330.13  5486.2  337.30  5559.0  345.68
  5594.7  346.91  5629.9  351.44  5727.7  358.40  5779.9  358.94  5810.8  360.30
#Mann=11,-1,0
  3211.4    0.05       0  3807.0    0.12       0  4020.3    0.05       0
  4098.2    0.03       0  4385.8    0.12       0  4456.3    0.05       0
  5306.0     0.1       0  5376.9    0.12       0  5486.2    0.05       0
  5727.7    0.12       0  5779.9    0.05       0
Bank Sta=4098.2,5376.9
Exp/Cntr=0.3,0.1

Type RM Length L Ch R = 1,28636,569,569,569
BEGIN DESCRIPTION:
Clear Creek 48.0
END DESCRIPTION:
XS GIS Cut Line= 3
      2741975.99      6782811.01      2741176.00      6784111.00
      2740869.45      6785110.63
#Sta/Elev= 30
  3473.9  381.35  3545.4  378.65  3555.0  375.67  3576.3  372.36  3582.1  372.73
  3597.5  369.43  3618.8  368.67  3655.5  364.61  3670.9  361.65  3676.8  362.74
  3713.5  359.65  3728.9  356.96  3850.7  343.44  3896.6  338.99  3914.2  338.94
  3939.5  335.42  3982.1  331.93  4012.9  330.82  4098.0  324.61  4282.4  322.00
  4285.0  321.50  5484.8  322.00  5490.8  322.00  5502.4  326.30  5648.8  345.14
  5697.7  348.73  5764.0  350.11  5866.7  352.41  6014.5  359.40  6045.9  361.20
#Mann=5,-1,0
  3473.9    0.05       0  4282.4    0.03       0  5484.8    0.05       0
  5764.0    0.12       0  6014.5    0.05       0
Bank Sta=4282.4,5484.8
Exp/Cntr=0.3,0.1

Type RM Length L Ch R = 1,28067,566,566,566
BEGIN DESCRIPTION:
Clear Creek 47.0
END DESCRIPTION:
XS GIS Cut Line= 3
      2740875.99      6782311.04      2740676.00      6783911.00
      2740576.00      6785161.00
#Sta/Elev= 30
  3383.1  383.18  3420.9  378.10  3443.5  376.79  3501.5  368.27  3506.5  369.02
  3524.1  366.96  3574.5  364.96  3582.1  365.01  3587.1  366.79  3711.2  364.79
  3786.2  357.91  3824.0  351.67  3846.6  351.93  3957.5  341.57  3990.2  341.23
  4007.9  337.75  4065.8  332.13  4070.9  332.84  4088.5  329.81  4159.3  325.35
  4192.2  323.79  4246.1  322.00  4248.8  321.50  5573.6  322.00  5617.5  322.45
  5806.8  340.59  6028.8  348.84  6161.8  359.01  6179.3  361.08  6249.5  363.53
#Mann=7,-1,0
  3383.1    0.12       0  3711.2    0.05       0  4159.3    0.12       0
  4192.2    0.05       0  4246.1    0.03       0  5573.6    0.05       0
  6161.8    0.12       0
Bank Sta=4246.1,5573.6
Exp/Cntr=0.3,0.1

Type RM Length L Ch R = 1,27501,598,598,598
BEGIN DESCRIPTION:
Clear Creek 46.0
END DESCRIPTION:
XS GIS Cut Line= 3
      2740775.98      6782561.04      2740126.00      6783861.00
      2740476.00      6785261.01
#Sta/Elev= 30
  3546.6  373.33  3605.3  371.63  3644.4  367.37  3650.0  368.16  3689.1  365.23
  3698.8  365.86  3711.5  365.07  3717.1  366.36  3733.8  365.72  3739.4  366.92
  3784.1  367.39  3806.5  365.68  3823.3  360.63  3828.9  361.06  3845.6  351.85
  3873.6  350.90  3889.5  347.65  3979.8  333.22  4056.2  325.16  4091.9  322.00
  4094.6  321.50  5845.8  322.00  5889.0  325.64  6048.8  335.07  6102.9  340.72
  6136.4  341.10  6144.2  343.64  6288.5  355.51  6378.7  365.10  6443.1  367.64
#Mann=6,-1,0
  3546.6    0.12       0  3698.8    0.05       0  3889.5    0.12       0
  4056.2    0.05       0  4091.9    0.03       0  5845.8    0.05       0
Bank Sta=4091.9,5845.8
Exp/Cntr=0.3,0.1

Type RM Length L Ch R = 1,26903,566,566,566
BEGIN DESCRIPTION:
Clear Creek 45.0
END DESCRIPTION:
XS GIS Cut Line= 3
      2740625.98      6782561.02      2739526.00      6783861.00
      2740326.02      6785261.04
#Sta/Elev= 30
  3301.2  372.95  3365.5  363.90  3372.0  361.88  3400.6  358.86  3407.2  357.25
  3414.9  357.13  3421.4  354.59  3464.3  347.83  3585.2  336.53  3620.3  331.44
  3650.9  331.21  3669.7  330.99  3698.3  327.16  3748.7  324.37  3776.3  323.25
  3798.4  323.80  3804.9  322.08  3812.0  322.00  3814.7  321.50  6199.1  322.00
  6213.4  322.15  6221.4  324.41  6264.6  327.15  6307.7  331.82  6366.8  336.24
  6432.3  344.33  6463.2  345.26  6469.0  347.64  6484.8  349.87  6616.6  366.46
#Mann=5,-1,0
  3301.2    0.12       0  3650.9     0.1       0  3748.7    0.05       0
  3812.0    0.03       0  6199.1    0.05       0
Bank Sta=3812,6199.1
Exp/Cntr=0.3,0.1

Type RM Length L Ch R = 1,26337,543,543,543
BEGIN DESCRIPTION:
Clear Creek 44.0
END DESCRIPTION:
XS GIS Cut Line= 3
      2740676.01      6782461.00      2739126.00      6783461.00
      2737526.00      6783961.00
#Sta/Elev= 30
  3155.4  380.20  3163.0  378.58  3168.9  379.53  3184.1  378.77  3199.3  376.05
  3220.4  375.36  3262.7  370.63  3293.0  364.76  3322.0  361.21  3344.5  355.56
  3365.6  352.11  3423.0  344.87  3478.3  340.03  3589.3  331.39  3604.5  329.08
  3749.7  324.01  3866.0  322.00  3868.7  321.50  6066.5  321.99  6106.6  322.00
  6131.5  326.12  6183.9  326.80  6300.4  336.23  6341.0  340.75  6362.5  340.93
  6406.8  346.80  6498.2  356.76  6526.4  358.66  6595.1  362.18  6676.3  363.66
#Mann=8,-1,0
  3155.4    0.12       0  3478.3     0.1       0  3866.0    0.03       0
  6066.5    0.12       0  6106.6     0.1       0  6300.4    0.05       0
  6406.8    0.12       0  6526.4    0.05       0
Bank Sta=3866,6106.6
Exp/Cntr=0.3,0.1

Type RM Length L Ch R = 1,25794,584,584,584
BEGIN DESCRIPTION:
Clear Creek 43.0
END DESCRIPTION:
XS GIS Cut Line= 3
      2740026.03      6782060.98      2738776.00      6783061.00
      2737475.96      6783861.02
#Sta/Elev= 30
  3398.8  359.64  3403.4  359.51  3455.7  354.96  3470.1  351.95  3493.7  349.83
  3532.6  344.78  3562.9  343.34  3662.2  332.41  3683.0  332.37  3691.0  329.83
  3711.8  328.99  3726.2  326.59  3748.0  326.03  3761.4  325.95  3769.4  323.63
  3790.5  322.00  3793.3  321.50  5955.3  321.99  5998.7  322.00  6009.4  322.00
  6017.9  324.88  6166.8  339.05  6207.2  343.29  6234.3  344.09  6290.1  350.59
  6304.3  351.85  6373.4  357.48  6396.5  361.07  6475.8  364.13  6526.1  363.72
#Mann=11,-1,0
  3398.8     0.1       0  3403.4    0.12       0  3493.7     0.1       0
  3532.6    0.12       0  3748.0    0.05       0  3790.5    0.03       0
  5955.3    0.12       0  5998.7    0.05       0  6166.8    0.05       0
  6290.1    0.12       0  6304.3    0.05       0
Bank Sta=3790.5,5998.7
Exp/Cntr=0.3,0.1

Type RM Length L Ch R = 1,25210,524,524,524
BEGIN DESCRIPTION:
Clear Creek 42.0
END DESCRIPTION:
XS GIS Cut Line= 3
      2740067.50      6781729.88      2738676.00      6782511.00
      2737525.99      6783761.01
#Sta/Elev= 30
  3408.4  380.67  3411.1  380.67  3451.6  375.43  3505.1  364.61  3521.1  358.91
  3533.7  357.53  3580.4  349.30  3607.8  347.35  3623.7  343.12  3651.2  341.46
  3673.9  337.62  3688.8  338.08  3726.4  334.22  3769.8  332.48  3795.0  328.94
  3796.6  328.75  3834.8  326.29  3843.2  322.00  3846.0  321.50  6216.2  322.00
  6237.2  322.00  6256.6  322.36  6270.8  325.46  6448.4  343.44  6476.1  344.45
  6490.3  347.93  6559.5  354.15  6591.3  357.16  6624.7  360.33  6702.7  363.13
#Mann=12,-1,0
  3408.4    0.05       0  3411.1    0.12       0  3451.6     0.1       0
  3533.7    0.12       0  3795.0     0.1       0  3796.6    0.05       0
  3843.2    0.03       0  6216.2    0.12       0  6237.2    0.05       0
  6448.4    0.05       0  6559.5    0.12       0  6591.3    0.05       0
Bank Sta=3843.2,6237.2
Exp/Cntr=0.3,0.1

Type RM Length L Ch R = 1,24686,565,565,565
BEGIN DESCRIPTION:
Clear Creek 41.0
END DESCRIPTION:
XS GIS Cut Line= 3
      2740039.64      6780918.75      2738476.00      6782061.00
      2737476.00      6783611.00
#Sta/Elev= 30
  3063.6  375.06  3110.6  371.81  3175.5  362.37  3204.3  359.83  3211.0  358.25
  3261.2  352.61  3382.5  342.19  3533.1  332.55  3648.1  330.31  3753.3  326.00
  3875.9  324.00  3890.6  323.95  3891.1  322.00  3893.9  321.50  6354.6  322.00
  6374.4  322.47  6380.5  324.02  6398.5  325.61  6404.1  325.86  6498.4  332.75
  6519.6  334.99  6525.5  336.93  6572.9  339.53  6628.5  344.11  6649.6  344.54
  6655.5  346.86  6701.1  351.12  6743.3  353.04  6815.9  358.69  6844.6  359.29
#Mann=8,-1,0
  3063.6     0.1       0  3753.3    0.12       0  3875.9    0.05       0
  3891.1    0.03       0  6354.6    0.05       0  6398.5     0.1       0
  6404.1    0.12       0  6572.9    0.05       0
Bank Sta=3891.1,6354.6
Exp/Cntr=0.3,0.1

Type RM Length L Ch R = 1,24121,563,563,563
BEGIN DESCRIPTION:
Clear Creek 40.0
END DESCRIPTION:
XS GIS Cut Line= 3
      2739426.02      6780310.98      2738176.00      6781611.00
      2736875.99      6783161.01
#Sta/Elev= 30
  3201.6  381.32  3258.1  383.52  3339.9  377.02  3378.5  375.24  3392.7  371.37
  3406.8  365.92  3427.9  362.85  3498.6  348.70  3661.2  332.99  3873.5  326.13
  3993.6  324.46  4000.8  324.17  4007.7  322.00  4010.5  321.50  6369.8  322.00
  6439.4  326.67  6468.5  330.59  6517.4  332.50  6605.3  339.43  6694.4  345.88
  6708.7  345.59  6786.8  350.58  6807.6  353.49  6864.8  356.91  6883.0  356.83
  6900.4  357.73  6942.9  358.16  6957.2  357.19  7020.9  360.32  7028.1  359.46
#Mann=8,-1,0
  3201.6    0.05       0  3339.9     0.1       0  4007.7    0.03       0
  6369.8     0.1       0  6468.5    0.12       0  6605.3     0.1       0
  6883.0    0.05       0  6900.4     0.1       0
Bank Sta=4007.7,6369.8
Exp/Cntr=0.3,0.1

Type RM Length L Ch R = 1,23558,543,543,543
BEGIN DESCRIPTION:
Clear Creek 39.0
END DESCRIPTION:
XS GIS Cut Line= 3
      2738676.02      6780310.98      2737976.00      6781111.00
      2736963.62      6782752.70
#Sta/Elev= 30
  3937.2  355.72  4015.5  341.01  4107.6  330.53  4114.2  330.90  4136.1  328.92
  4192.1  326.26  4199.7  322.00  4202.5  321.50  4235.1  321.50  6511.4  322.00
  6522.8  322.03  6533.7  322.40  6539.5  325.27  6576.2  327.49  6585.7  326.78
  6607.0  329.13  6612.9  331.50  6628.3  332.20  6670.8  337.20  6701.6  338.70
  6707.5  340.28  6722.9  341.50  6728.8  343.26  6748.2  345.21  6780.9  348.69
  6786.7  350.29  6832.9  352.96  6844.8  354.67  6896.8  356.67  6929.0  356.59
#Mann=6,-1,0
  3937.2     0.1       0  4199.7    0.03       0  4235.1    0.05       0
  6511.4     0.1       0  6522.8    0.12       0  6748.2    0.05       0
Bank Sta=4199.7,6511.4
Exp/Cntr=0.3,0.1

Type RM Length L Ch R = 1,23015,566,566,566
BEGIN DESCRIPTION:
Clear Creek 38.0
END DESCRIPTION:
XS GIS Cut Line= 3
      2738513.29      6779822.80      2737576.00      6780761.00
      2736874.52      6782717.68
#Sta/Elev= 30
  3673.9  373.33  3713.1  369.94  3776.8  360.39  3790.9  361.31  3812.1  360.59
  3854.6  351.41  3925.3  343.85  3939.4  339.88  3974.8  338.46  4024.3  331.88
  4073.6  328.63  4172.8  325.55  4204.1  322.72  4215.0  322.00  4217.8  321.50
  6440.6  322.00  6475.4  323.80  6508.6  323.52  6525.3  325.06  6581.5  325.38
  6617.6  327.33  6657.3  331.22  6699.2  333.14  6735.3  336.97  6760.7  338.00
  6796.8  342.33  6847.6  346.32  6873.8  350.36  6939.9  356.15  7078.7  357.37
#Mann=7,-1,0
  3673.9    0.05       0  4073.6    0.12       0  4204.1    0.05       0
  4215.0    0.03       0  6440.6    0.05       0  6475.4    0.12       0
  6873.8    0.05       0
Bank Sta=4215,6440.6
Exp/Cntr=0.3,0.1

Type RM Length L Ch R = 1,22449,600,600,600
BEGIN DESCRIPTION:
Clear Creek 37.0
END DESCRIPTION:
XS GIS Cut Line= 3
      2736926.00      6779261.04      2737026.00      6780711.00
      2736826.00      6782711.02
#Sta/Elev= 30
  3546.6  383.97  3586.2  381.96  3615.5  378.97  3620.5  380.28  3656.8  377.40
  3781.3  364.70  4017.7  344.79  4027.7  342.48  4181.6  332.79  4288.3  326.54
  4332.1  322.06  4335.3  322.00  4338.1  321.50  5775.2  322.00  5793.9  322.00
  5814.0  325.02  5952.2  333.34  6052.7  334.73  6075.3  336.45  6343.1  330.72
  6386.9  331.45  6396.9  330.09  6407.0  325.95  6427.1  331.92  6441.3  331.64
  6628.1  338.41  6720.6  345.49  6735.9  346.52  6856.7  352.91  7010.0  356.44
#Mann=11,-1,0
  3546.6    0.05       0  3586.2     0.1       0  3781.3    0.05       0
  4181.6    0.12       0  4332.1    0.05       0  4335.3    0.03       0
  5775.2    0.05       0  6343.1    0.12       0  6441.3    0.05       0
  6720.6    0.12       0  6735.9    0.05       0
Bank Sta=4335.3,5775.2
Exp/Cntr=0.3,0.1

Type RM Length L Ch R = 1,21849,568,568,568
BEGIN DESCRIPTION:
Clear Creek 36.0
END DESCRIPTION:
XS GIS Cut Line= 3
      2736626.00      6779411.00      2736426.00      6780711.00
      2736476.00      6782111.01
#Sta/Elev= 30
  3684.7  379.57  3713.8  376.60  3718.8  377.72  3765.6  371.36  3782.1  367.20
  3806.1  366.77  3836.5  362.08  3867.7  359.36  3907.3  354.08  3937.6  353.44
  3957.9  349.16  4018.6  341.43  4065.2  338.31  4089.4  335.52  4108.4  335.07
  4140.0  330.74  4163.9  330.01  4250.6  324.53  4277.3  322.00  4280.2  321.50
  5961.4  322.00  5970.6  325.43  5978.1  326.45  6050.7  330.62  6100.7  336.44
  6150.7  339.76  6190.8  344.19  6240.8  345.26  6280.8  349.25  6400.9  350.04
#Mann=7,-1,0
  3684.7    0.05       0  3867.7    0.12       0  4065.2    0.05       0
  4163.9    0.12       0  4250.6    0.05       0  4277.3    0.03       0
  5961.4    0.05       0
Bank Sta=4277.3,5961.4
Exp/Cntr=0.3,0.1

Type RM Length L Ch R = 1,21281,566,566,566
BEGIN DESCRIPTION:
Clear Creek 35.0
END DESCRIPTION:
XS GIS Cut Line= 3
      2736382.13      6779446.75      2735876.00      6780661.00
      2735926.00      6781910.98
#Sta/Elev= 30
  3684.1  367.89  3690.6  366.65  3743.7  362.97  3767.5  359.68  3820.6  356.03
  3897.5  354.58  3905.4  351.84  3945.1  349.62  4044.4  341.28  4098.9  335.17
  4128.2  333.78  4133.6  332.17  4152.0  332.59  4157.4  326.82  4175.8  328.85
  4181.3  323.83  4193.4  324.32  4205.1  324.78  4210.5  322.36  4226.8  322.00
  4229.6  321.50  5953.7  322.00  5960.4  322.00  5970.4  326.77  6060.5  335.97
  6090.5  341.79  6100.5  342.77  6170.6  345.92  6210.6  350.19  6250.6  350.78
#Mann=5,-1,0
  3684.1    0.05       0  4044.4    0.12       0  4193.4    0.05       0
  4226.8    0.03       0  5953.7    0.05       0
Bank Sta=4226.8,5953.7
Exp/Cntr=0.3,0.1

Type RM Length L Ch R = 1,20715,566,566,566
BEGIN DESCRIPTION:
Clear Creek 34.0
END DESCRIPTION:
XS GIS Cut Line= 3
      2736331.44      6779348.61      2735476.00      6780261.00
      2734776.02      6781660.96
#Sta/Elev= 30
  3749.3  364.14  3861.1  357.72  3938.8  351.36  3945.7  350.21  3953.0  345.55
  3967.2  344.19  3974.0  346.20  3988.2  345.88  4044.8  340.89  4080.5  339.51
  4115.6  335.18  4306.3  322.00  4309.1  321.50  5858.1  322.00  5859.5  322.00
  5880.4  322.00  5886.0  328.01  5925.2  327.69  6037.0  330.95  6064.9  334.54
  6115.4  335.09  6193.5  338.66  6221.4  341.96  6260.6  341.71  6266.2  343.65
  6288.5  345.44  6305.3  343.19  6333.3  346.31  6417.1  346.72  6565.2  351.57
#Mann=5,-1,0
  3749.3    0.05       0  4306.3    0.03       0  5858.1    0.12       0
  5859.5    0.05       0  6115.4    0.05       0
Bank Sta=4306.3,5859.5
Exp/Cntr=0.3,0.1

Type RM Length L Ch R = 1,20149,581,581,581
BEGIN DESCRIPTION:
Clear Creek 33.0
END DESCRIPTION:
XS GIS Cut Line= 3
      2736340.95      6779196.41      2735076.00      6779861.00
      2734686.36      6781200.89
#Sta/Elev= 30
  3571.1  368.48  3696.6  358.95  3719.3  356.47  3725.0  357.20  3734.8  354.97
  3741.3  355.58  3807.5  349.95  3836.5  346.29  3873.6  344.01  3912.1  339.75
  3961.8  336.89  3969.0  335.06  3978.2  333.00  4044.4  331.57  4066.4  329.97
  4082.8  327.32  4164.1  323.62  4178.5  322.00  4181.4  321.50  5880.5  322.00
  5895.6  323.86  5917.4  328.75  5945.8  332.50  5984.5  335.96  6023.2  337.33
  6090.3  342.06  6228.9  348.41  6240.0  347.57  6301.8  348.48  6395.4  347.96
#Mann=5,-1,0
  3571.1    0.05       0  3696.6     0.1       0  3969.0    0.05       0
  4178.5    0.03       0  5880.5    0.05       0
Bank Sta=4178.5,5880.5
Exp/Cntr=0.3,0.1

Type RM Length L Ch R = 1,19568,563,563,563
BEGIN DESCRIPTION:
Clear Creek 32.0
END DESCRIPTION:
XS GIS Cut Line= 3
      2735126.00      6778211.00      2734626.00      6779511.00
      2734592.39      6781191.72
#Sta/Elev= 30
  3602.2  357.89  3687.6  357.98  3731.8  357.78  3781.9  356.28  3841.1  354.36
  3912.9  350.41  3980.4  345.76  3998.6  344.05  4010.4  341.75  4035.1  341.74
  4065.1  340.08  4095.1  336.52  4137.9  332.04  4144.3  330.43  4199.1  325.72
  4245.1  324.03  4251.9  322.00  4254.8  321.50  6168.2  322.00  6195.3  322.56
  6210.3  324.73  6235.3  326.67  6242.9  327.97  6265.3  328.25  6415.3  337.03
  6495.3  340.22  6505.3  339.74  6565.7  342.62  6647.8  346.22  6676.1  347.45
#Mann=10,-1,0
  3602.2    0.05       0  3687.6    0.12       0  3781.9    0.05       0
  4095.1    0.12       0  4199.1    0.05       0  4251.9    0.03       0
  6168.2    0.05       0  6210.3     0.1       0  6565.7    0.05       0
  6647.8     0.1       0
Bank Sta=4251.9,6168.2
Exp/Cntr=0.3,0.1

Type RM Length L Ch R = 1,19005,585,585,585
BEGIN DESCRIPTION:
Clear Creek 31.0
END DESCRIPTION:
XS GIS Cut Line= 3
      2734975.97      6778411.03      2734176.00      6779211.00
      2733576.00      6781011.00
#Sta/Elev= 30
  3868.7  352.59  3896.9  351.12  3995.9  343.56  4030.1  342.54  4066.7  339.54
  4094.9  335.60  4123.2  333.20  4173.5  326.31  4193.9  324.35  4207.7  322.00
  4210.5  321.50  5858.6  322.00  5864.4  324.17  5927.6  323.63  5990.9  325.03
  6138.5  328.95  6159.5  330.86  6191.2  330.92  6296.6  334.94  6380.9  336.48
  6402.0  337.82  6412.5  339.65  6444.1  341.05  6465.2  340.92  6486.3  341.88
  6517.9  341.31  6623.3  343.17  6644.4  344.66  6855.2  351.32  6897.4  350.94
#Mann=5,-1,0
  3868.7    0.05       0  4030.1    0.12       0  4173.5    0.05       0
  4207.7    0.03       0  5858.6    0.05       0
Bank Sta=4207.7,5858.6
Exp/Cntr=0.3,0.1

Type RM Length L Ch R = 1,18420,542,542,542
BEGIN DESCRIPTION:
Clear Creek 30.0
END DESCRIPTION:
XS GIS Cut Line= 3
      2734976.00      6777561.00      2733726.00      6778861.00
      2733526.00      6780660.96
#Sta/Elev= 30
  3201.3  384.02  3271.9  384.86  3300.2  384.03  3336.2  380.50  3427.6  373.74
  3434.8  371.31  3448.9  370.30  3505.5  367.49  3519.7  368.16  3544.7  365.82
  3554.9  366.35  3569.1  363.57  3604.3  362.30  3675.1  356.26  3717.5  350.55
  3738.9  350.05  3775.4  344.44  3777.9  344.18  3866.2  333.81  3910.7  330.38
  3921.8  329.69  3958.1  326.16  3965.0  322.65  3978.7  322.00  3981.6  321.50
  6065.0  322.00  6081.3  324.43  6151.8  326.49  6463.7  332.16  6815.8  347.08
#Mann=9,-1,0
  3201.3    0.05       0  3336.2    0.12       0  3544.7    0.05       0
  3775.4    0.12       0  3777.9    0.05       0  3910.7    0.12       0
  3921.8    0.05       0  3978.7    0.03       0  6065.0    0.05       0
Bank Sta=3978.7,6065
Exp/Cntr=0.3,0.1

Type RM Length L Ch R = 1,17878,548,548,548
BEGIN DESCRIPTION:
Clear Creek 29.0
END DESCRIPTION:
XS GIS Cut Line= 3
      2734826.01      6777610.99      2733276.00      6778611.00
      2733476.00      6780811.03
#Sta/Elev= 30
  3155.4  376.34  3163.0  374.93  3220.4  372.37  3257.5  368.02  3262.7  368.81
  3314.1  366.06  3329.3  363.17  3371.6  360.81  3401.9  356.06  3429.1  355.05
  3438.2  353.10  3444.6  353.85  3459.3  350.50  3642.1  334.08  3683.1  330.86
  3726.6  325.53  3740.5  322.47  3756.3  322.00  3759.1  321.50  6269.2  322.00
  6285.3  325.79  6315.4  327.19  6466.0  329.50  6476.1  324.56  6486.1  322.87
  6506.2  328.01  6516.2  328.65  6686.9  332.08  7008.2  345.64  7209.1  350.43
#Mann=6,-1,0
  3155.4    0.12       0  3257.5    0.05       0  3444.6    0.12       0
  3642.1    0.05       0  3756.3    0.03       0  6269.2    0.05       0
Bank Sta=3756.3,6269.2
Exp/Cntr=0.3,0.1

Type RM Length L Ch R = 1,17330,565,565,565
BEGIN DESCRIPTION:
Clear Creek 28.0
END DESCRIPTION:
XS GIS Cut Line= 4
      2734326.01      6777460.99      2732776.00      6778461.00
      2731374.29      6779862.64      2730547.05      6779996.07
#Sta/Elev= 30
  3155.4  350.61  3190.8  349.68  3214.5  349.29  3220.4  348.01  3235.6  347.79
  3256.7  345.89  3277.8  341.99  3293.0  341.24  3314.4  337.31  3322.0  336.10
  3329.3  333.27  3386.7  329.14  3393.4  327.46  3423.0  325.24  3443.8  322.00
  3446.8  321.40  7088.7  322.00  7102.1  322.26  7112.2  324.82  7190.0  335.11
  7195.0  334.88  7256.8  340.94  7264.2  342.50  7304.7  344.27  7313.5  346.52
  7324.9  347.68  7442.2  351.94  7509.0  352.22  7632.6  354.90  7820.2  361.97
#Mann=5,-1,0
  3155.4    0.12       0  3190.8    0.05       0  3314.4    0.12       0
  3443.8    0.03       0  7088.7    0.05       0
Bank Sta=3443.8,7088.7
Exp/Cntr=0.3,0.1

Type RM Length L Ch R = 1,16765,566,566,566
BEGIN DESCRIPTION:
Clear Creek 27.0
END DESCRIPTION:
XS GIS Cut Line= 3
      2733926.02      6776460.98      2732376.00      6778061.00
      2730926.00      6779611.00
#Sta/Elev= 30
  2772.3  354.63  2836.0  353.07  2871.3  349.71  2949.2  343.88  2970.3  344.36
  2977.5  342.94  3048.2  336.01  3081.0  334.16  3097.6  333.36  3140.1  328.68
  3182.5  326.50  3188.3  322.00  3191.3  321.40  6578.0  322.00  6604.4  322.00
  6641.6  322.00  6648.4  323.30  6655.7  325.76  6726.1  331.42  6825.3  337.44
  6860.9  338.85  6865.5  338.29  6875.1  338.51  6881.9  340.31  6889.2  339.66
  6896.1  341.58  6931.3  343.91  7030.4  347.99  7066.1  350.23  7122.5  350.65
#Mann=6,-1,0
  2772.3    0.05       0  3081.0    0.12       0  3188.3    0.03       0
  6578.0    0.12       0  6604.4    0.12       0  6865.5    0.05       0
Bank Sta=3188.3,6604.4
Exp/Cntr=0.3,0.1

Type RM Length L Ch R = 1,16199,567,567,567
BEGIN DESCRIPTION:
Clear Creek 26.0
END DESCRIPTION:
XS GIS Cut Line= 3
      2733526.02      6776060.98      2731976.00      6777661.00
      2730375.99      6779861.01
#Sta/Elev= 30
  2772.3  359.65  2984.4  352.03  3175.5  349.35  3224.9  346.14  3314.2  334.30
  3343.6  332.62  3423.0  324.99  3472.4  324.71  3485.2  322.00  3488.2  321.40
  6678.3  321.99  6716.9  322.00  6746.2  322.00  6754.7  325.54  6811.1  326.11
  6825.8  329.13  6852.0  329.71  6961.8  332.92  7047.6  332.07  7148.0  336.91
  7176.2  341.02  7254.7  345.55  7304.9  346.80  7319.6  344.99  7334.3  345.61
  7340.5  348.15  7376.0  347.21  7434.7  352.62  7584.3  361.02  7720.3  366.06
#Mann=7,-1,0
  2772.3    0.05       0  3314.2    0.12       0  3343.6    0.05       0
  3485.2    0.03       0  6678.3    0.12       0  6716.9    0.05       0
  6852.0    0.05       0
Bank Sta=3485.2,6716.9
Exp/Cntr=0.3,0.1

Type RM Length L Ch R = 1,15632,1077,1077,1077
BEGIN DESCRIPTION:
Clear Creek 25.0
END DESCRIPTION:
XS GIS Cut Line= 3
      2732854.93      6775756.69      2731576.00      6777261.00
      2730242.94      6779256.15
#Sta/Elev= 30
  3030.5  329.69  3061.6  326.66  3082.5  327.20  3089.1  329.63  3096.8  327.07
  3103.3  330.80  3139.6  326.32  3174.7  331.29  3203.3  331.58  3238.4  327.19
  3281.3  331.69  3330.7  330.76  3345.0  334.15  3373.5  335.58  3394.4  333.30
  3437.2  335.55  3510.4  333.54  3600.6  332.22  3667.6  325.79  3719.3  322.00
  3722.3  321.30  6613.3  321.99  6659.4  322.00  6670.3  325.24  6758.3  331.40
  6857.1  340.21  6979.7  347.35  7096.8  347.04  7268.0  356.71  7404.5  361.30
#Mann=7,-1,0
  3030.5    0.05       0  3510.4    0.12       0  3667.6    0.05       0
  3719.3    0.03       0  6613.3    0.12       0  6659.4    0.05       0
  6758.3    0.05       0
Bank Sta=3719.3,6659.4
Exp/Cntr=0.3,0.1

Type RM Length L Ch R = 1,14555,738,738,738
BEGIN DESCRIPTION:
Clear Creek 24.0
END DESCRIPTION:
XS GIS Cut Line= 3
      2732299.57      6774726.19      2731176.00      6776311.00
      2730133.67      6778810.05
#Sta/Elev= 30
  3050.8  342.13  3156.5  341.68  3228.3  336.85  3307.8  335.19  3314.1  333.64
  3361.6  330.35  3423.5  327.38  3429.6  326.82  3439.1  324.27  3444.4  323.95
  3449.8  322.00  3452.8  321.30  7012.0  322.00  7028.2  322.00  7041.3  322.23
  7063.5  327.09  7073.8  327.11  7105.8  329.43  7111.2  330.71  7171.3  334.53
  7218.9  336.75  7279.7  339.27  7294.2  341.62  7365.7  346.83  7377.2  348.58
  7448.0  354.27  7524.9  355.95  7601.8  359.27  7678.7  360.51  7701.2  362.74
#Mann=7,-1,0
  3050.8    0.05       0  3361.6    0.12       0  3439.1    0.05       0
  3449.8    0.03       0  7012.0    0.12       0  7028.2    0.05       0
  7218.9    0.05       0
Bank Sta=3449.8,7028.2
Exp/Cntr=0.3,0.1

Type RM Length L Ch R = 1,13817,327,327,327
BEGIN DESCRIPTION:
Clear Creek 23.0
END DESCRIPTION:
XS GIS Cut Line= 3
      2731124.02      6774244.01      2730625.86      6775861.33
      2729912.71      6778426.02
#Sta/Elev= 30
  3307.7  335.87  3440.6  325.59  3525.7  324.05  3529.7  322.00  3532.7  321.30
  6530.1  321.99  6585.6  322.00  6598.1  324.48  6697.3  325.56  6731.5  326.72
  6743.4  328.55  6770.9  327.46  6776.1  329.59  6810.4  331.04  6857.6  330.49
  6878.3  335.04  6918.2  334.01  6962.9  338.14  6997.1  336.87  7002.9  335.34
  7031.3  336.82  7036.5  339.75  7044.4  340.38  7117.6  340.91  7178.6  342.98
  7223.2  348.18  7365.4  349.81  7428.4  352.47  7444.2  354.48  7662.0  359.37
#Mann=5,-1,0
  3307.7    0.05       0  3529.7    0.03       0  6530.1    0.12       0
  6585.6    0.05       0  7117.6    0.05       0
Bank Sta=3529.7,6585.6
Exp/Cntr=0.3,0.1

Type RM Length L Ch R = 1,13490,621,621,621
BEGIN DESCRIPTION:
Clear Creek 22.0
END DESCRIPTION:
XS GIS Cut Line= 4
      2730737.57      6774245.72      2730331.18      6775760.56
      2729658.38      6778071.30      2729602.23      6778595.51
#Sta/Elev= 30
  3431.6  340.25  3494.8  335.90  3503.1  336.31  3649.6  327.02  3664.8  328.54
  3684.4  325.29  3737.3  323.70  3742.5  322.00  3745.5  321.30  3819.0  321.31
  6550.5  321.94  6778.1  321.99  6828.6  322.00  6854.4  322.00  6860.2  325.90
  6865.4  323.27  6875.2  326.35  6932.4  327.60  6965.9  330.05  7043.3  331.29
  7110.3  334.87  7281.4  339.15  7394.0  344.83  7571.1  348.73  7627.7  351.53
  7663.3  352.47  7668.3  351.72  7755.5  355.34  7847.7  356.99  7933.9  356.35
#Mann=7,-1,0
  3431.6    0.05       0  3503.1    0.12       0  3742.5    0.05       0
  3819.0    0.05       0  6550.5   0.075       0  6778.1    0.05       0
  6828.6    0.12       0
Bank Sta=3742.5,6828.6
Exp/Cntr=0.3,0.1

Type RM Length L Ch R = 1,12869,600,600,600
BEGIN DESCRIPTION:
Clear Creek 21.0
END DESCRIPTION:
XS GIS Cut Line= 4
      2730207.18      6774390.96      2729726.00      6775711.00
      2729150.20      6778019.99      2729545.54      6778746.25
#Sta/Elev= 30
  3595.0  343.50  3728.7  340.44  3815.3  336.96  3864.2  331.27  3925.0  324.15
  3930.8  322.00  3933.8  321.30  7200.5  322.00  7210.9  323.30  7216.0  322.16
  7226.2  323.70  7257.3  325.47  7308.6  326.34  7415.0  324.79  7422.0  325.65
  7503.6  326.80  7591.0  335.21  7656.6  337.01  7665.5  338.31  7700.2  339.73
  7745.2  340.71  7760.1  339.99  7879.8  345.22  7916.0  347.69  7945.3  347.77
  8070.6  352.08  8130.5  352.35  8158.0  353.70  8174.2  353.05  8206.6  354.54
#Mann=5,-1,0
  3595.0    0.05       0  3728.7    0.12       0  3864.2    0.05       0
  3930.8    0.03       0  7200.5    0.05       0
Bank Sta=3930.8,7200.5
Exp/Cntr=0.3,0.1
