--- Dry Creek.prj (project) ---

Proj Title=Dry Creek Base Level Engineering
Current Plan=p01
Default Exp/Contr=0.3,0.1
English Units
Geom File=g01
Flow File=f01
Plan File=p01
BEGIN DESCRIPTION:
Dry Creek
END DESCRIPTION:

--- Dry Creek.p01 (plan) ---

Plan Title=Multiple Run
Short Identifier=Multiple
Geom File=g01
Flow File=f01
Subcritical Flow
K Sum by GR= 0
Std Step Tol= 0.01
Critical Tol= 0.01
Num of Std Step Trials= 20
Max Error Tol= 0.3
Flow Tol Ratio= 0.001
Split Flow NTrial= 30
Split Flow Tol= 0.02
Split Flow Ratio= 0.02
Log Output Level= 0
Friction Slope Method= 1
Unsteady Friction Slope Method= 2
Unsteady Bridges Friction Slope Method= 1
Parabolic Critical Depth
Global Vel Dist=  1 , 1 , 1
Global Log Level= 0
CheckData=True
Encroach Param= -1, 0, 0, 0
BEGIN DESCRIPTION:
Multiple Run
END DESCRIPTION:

--- Dry Creek.f01 (steady flow) ---

Flow Title=Multiple
Number of Profiles=7
Profile Names=10-year,25-year,50-year,1pct_min,100-year,1pct_plu,500-year
River Rch & RM= Dry Creek,Reach-1,36269
     510     668     793     466     930    1856    1280
River Rch & RM= Dry Creek,Reach-1,32684
     993    1350    1642     988    1971    3932    2840
River Rch & RM= Dry Creek,Reach-1,23892
    1617    2249    2778    1694    3381    6745    5010
River Rch & RM= Dry Creek,Reach-1,22826
    1852    2593    3215    1968    3927    7836    5864
River Rch & RM= Dry Creek,Reach-1,16201
    1860    2607    3234    1981    3953    7887    5908
River Rch & RM= Dry Creek,Reach-1,14499
    1994    2800    3479    2133    4256    8491    6374
River Rch & RM= Dry Creek,Reach-1,11071
    2103    2954    3671    2251    4491    8960    6726
River Rch & RM= Dry Creek,Reach-1,8625
    2211    3108    3863    2369    4726    9430    7079
Boundary for River Rch & Prof#=Dry Creek,Reach-1,1
Up Type=0
Dn Type=3
Dn Slope=0.005
Boundary for River Rch & Prof#=Dry Creek,Reach-1,2
Up Type=0
Dn Type=3
Dn Slope=0.005
Boundary for River Rch & Prof#=Dry Creek,Reach-1,3
Up Type=0
Dn Type=3
Dn Slope=0.005
Boundary for River Rch & Prof#=Dry Creek,Reach-1,4
Up Type=0
Dn Type=3
Dn Slope=0.005
Boundary for River Rch & Prof#=Dry Creek,Reach-1,5
Up Type=0
Dn Type=3
Dn Slope=0.005
Boundary for River Rch & Prof#=Dry Creek,Reach-1,6
Up Type=0
Dn Type=3
Dn Slope=0.005
Boundary for River Rch & Prof#=Dry Creek,Reach-1,7
Up Type=0
Dn Type=3
Dn Slope=0.005

--- Dry Creek.g01 (geometry) ---

Geom Title=Existing Conditions

River Reach=Dry Creek,Reach-1
Reach XY= 30
      2737126.00      6849811.00      2735928.38      6847505.47
      2735725.55      6846521.19      2736126.10      6844740.90
      2735777.20      6844351.41      2735924.95      6843570.49
      2734927.97      6841005.64      2734922.46      6840312.46
      2734628.09      6840055.74      2734722.49      6839412.25
      2734078.17      6838505.55      2734122.45      6837862.47
      2733481.08      6837263.28      2733517.52      6836814.31
      2732936.27      6837060.02      2732131.58      6836605.42
      2731470.58      6834858.25      2731031.42      6834705.82
      2730579.27      6834059.66      2730515.05      6833100.98
      2729727.97      6832655.32      2729625.61      6831179.47
      2729876.56      6830883.83      2729575.64      6830435.80
      2729826.30      6828933.76      2729433.56      6827861.00
      2729726.45      6826884.06      2729527.13      6825270.44
      2729876.61      6824983.71      2729376.00      6822711.00

Type RM Length L Ch R = 1,36269,370,370,370
BEGIN DESCRIPTION:
Dry Creek36268.899
END DESCRIPTION:
XS GIS Cut Line= 3
      2737797.48      6849661.00      2737126.03      6849728.12
      2736662.72      6849761.36
#Sta/Elev= 30
  4325.2  460.95  4356.8  460.46  4427.2  458.90  4457.3  458.52  4547.8  456.40
  4567.9  456.20  4579.8  455.59  4668.4  454.00  4688.5  453.24  4748.8  452.17
  4758.8  451.73  4775.8  451.37  4780.8  451.44  4876.3  449.49  4881.3  449.67
  4919.6  449.14  4949.8  448.65  4959.8  448.26  4995.5  448.10  4995.8  447.60
  4999.3  447.60  4999.5  448.10  5010.1  448.27  5030.1  448.17  5050.2  448.55
  5200.5  451.93  5240.6  453.24  5350.9  456.23  5421.1  458.52  5464.5  459.68
#Mann=3,-1,0
  4325.2    0.05       0  4995.5    0.05       0  4999.5    0.05       0
Bank Sta=4995.5,4999.5
Exp/Cntr=0.3,0.1

Type RM Length L Ch R = 1,35899,291,291,291
BEGIN DESCRIPTION:
Dry Creek35899.11
END DESCRIPTION:
XS GIS Cut Line= 3
      2737459.20      6849154.22      2737048.41      6849383.45
      2736630.57      6849648.62
#Sta/Elev= 30
  4529.8  459.87  4558.0  459.22  4579.8  458.23  4633.4  456.55  4639.2  456.12
  4655.1  455.78  4682.6  454.62  4692.8  454.51  4705.2  453.84  4728.1  453.30
  4736.3  452.78  4751.0  452.50  4779.7  451.35  4860.8  449.19  4957.2  447.50
  4969.4  446.61  4996.7  446.36  4997.0  445.86  5000.5  445.86  5000.7  446.36
  5028.2  446.39  5043.4  447.53  5079.8  448.34  5116.3  449.49  5180.7  450.38
  5267.9  452.61  5392.4  455.14  5434.8  456.35  5441.3  456.76  5495.1  458.56
#Mann=3,-1,0
  4529.8    0.05       0  4996.7    0.05       0  5000.7    0.05       0
Bank Sta=4996.7,5000.7
Exp/Cntr=0.3,0.1

Type RM Length L Ch R = 1,35608,292,292,292
BEGIN DESCRIPTION:
Dry Creek35607.92
END DESCRIPTION:
XS GIS Cut Line= 3
      2737401.71      6849010.18      2736937.72      6849127.34
      2736576.80      6849482.47
#Sta/Elev= 30
  4526.1  460.27  4589.7  458.38  4594.9  458.55  4635.9  457.44  4677.0  456.14
  4738.3  453.87  4753.9  452.76  4759.1  452.95  4789.8  451.34  4795.0  451.44
  4810.5  450.47  4836.0  449.59  4841.4  449.18  4882.7  447.93  4923.9  447.04
  4944.5  445.91  4998.2  445.52  4998.5  445.02  5002.0  445.02  5002.2  445.52
  5029.7  445.67  5079.1  447.94  5114.5  448.89  5149.8  449.21  5171.1  448.77
  5185.3  448.79  5234.7  449.21  5397.4  452.52  5482.3  454.68  5511.0  455.72
#Mann=3,-1,0
  4526.1    0.05       0  4998.2    0.05       0  5002.2    0.05       0
Bank Sta=4998.2,5002.2
Exp/Cntr=0.3,0.1

Type RM Length L Ch R = 1,35316,388,388,388
BEGIN DESCRIPTION:
Dry Creek35315.61
END DESCRIPTION:
XS GIS Cut Line= 3
      2737177.80      6848540.77      2736778.32      6848912.28
      2736371.86      6849453.39
#Sta/Elev= 30
  4457.2  459.42  4494.0  458.55  4593.2  455.09  4635.7  453.48  4649.9  452.51
  4691.9  450.75  4784.3  447.84  4869.3  445.61  4897.1  445.23  4925.4  444.16
  4994.3  443.82  4994.5  443.32  4998.0  443.32  4998.3  443.82  5005.1  443.83
  5017.4  444.55  5032.0  444.48  5096.6  447.47  5145.0  448.56  5175.7  448.79
  5231.9  447.86  5256.4  448.12  5288.8  448.36  5331.9  449.67  5375.7  450.09
  5417.3  451.23  5531.9  453.02  5625.6  455.46  5631.9  455.26  5679.5  456.41
#Mann=5,-1,0
  4457.2    0.05       0  4994.3    0.05       0  4998.3    0.05       0
  5145.0   0.045       0  5256.4    0.05       0
Bank Sta=4994.3,4998.3
Exp/Cntr=0.3,0.1

Type RM Length L Ch R = 1,34928,387,387,387
BEGIN DESCRIPTION:
Dry Creek34928.33
END DESCRIPTION:
XS GIS Cut Line= 3
      2736971.70      6848314.20      2736630.69      6848572.82
      2735950.29      6848930.35
#Sta/Elev= 30
  4577.4  456.22  4714.6  452.55  4829.0  448.24  4864.3  446.19  4899.7  442.98
  4928.8  443.42  4943.3  442.92  4972.4  443.54  4978.7  442.75  4984.2  442.70
  4984.4  442.20  4987.9  442.20  4988.2  442.70  4988.8  442.80  4993.3  443.52
  5005.2  442.74  5014.3  443.39  5022.0  443.12  5036.3  443.55  5081.2  442.99
  5089.8  442.82  5103.7  444.41  5191.4  447.32  5251.1  447.73  5339.3  446.21
  5349.6  445.59  5355.7  444.22  5361.4  444.24  5438.2  446.43  5774.0  453.58
#Mann=6,-1,0
  4577.4    0.05       0  4984.2   0.045       0  4988.2    0.05       0
  4988.8   0.045       0  5081.2    0.05       0  5103.7   0.045       0
Bank Sta=4984.2,4988.2
Exp/Cntr=0.3,0.1

Type RM Length L Ch R = 1,34541,405,405,405
BEGIN DESCRIPTION:
Dry Creek34541.44
END DESCRIPTION:
XS GIS Cut Line= 3
      2736815.93      6847946.81      2736361.12      6848296.27
      2735897.51      6848645.52
#Sta/Elev= 30
  4426.5  453.62  4443.5  453.47  4478.8  452.22  4507.8  453.02  4514.7  451.91
  4522.3  451.52  4636.5  448.51  4665.5  448.06  4671.8  448.11  4678.6  448.78
  4692.7  448.44  4700.9  447.46  4750.7  445.85  4829.6  445.02  4835.9  445.33
  4879.4  444.93  4885.7  445.36  4921.1  444.41  4935.6  443.20  4962.6  442.67
  4962.8  442.17  4966.3  442.17  4966.6  442.67  5059.2  443.08  5129.0  443.21
  5135.3  442.68  5164.4  443.68  5285.2  445.61  5407.1  448.60  5580.5  453.59
#Mann=4,-1,0
  4426.5    0.05       0  4962.6    0.05       0  4966.6    0.05       0
  5059.2   0.045       0
Bank Sta=4962.6,4966.6
Exp/Cntr=0.3,0.1

Type RM Length L Ch R = 1,34136,340,340,340
BEGIN DESCRIPTION:
Dry Creek34135.81
END DESCRIPTION:
XS GIS Cut Line= 3
      2736646.93      6847641.47      2736172.13      6847966.21
      2735785.32      6848299.92
#Sta/Elev= 30
  4431.1  453.26  4453.6  452.86  4474.6  453.31  4489.5  452.52  4495.6  451.76
  4546.4  450.01  4576.2  449.56  4589.7  450.29  4612.1  448.28  4648.0  447.13
  4698.8  446.44  4797.6  443.08  4831.5  442.66  4831.7  442.16  4835.2  442.16
  4835.5  442.66  4869.3  443.26  4899.2  442.87  5048.5  442.89  5078.2  442.71
  5148.4  444.00  5283.4  447.44  5347.0  449.36  5354.7  449.99  5361.3  449.78
  5368.9  451.29  5375.5  450.26  5383.2  450.56  5389.8  450.09  5517.2  452.95
#Mann=4,-1,0
  4431.1    0.05       0  4831.5    0.05       0  4835.5    0.05       0
  5048.5   0.045       0
Bank Sta=4831.5,4835.5
Exp/Cntr=0.3,0.1

Type RM Length L Ch R = 1,33796,109,109,109
BEGIN DESCRIPTION:
Dry Creek33796.32
END DESCRIPTION:
XS GIS Cut Line= 3
      2736504.50      6847451.10      2735996.58      6847688.43
      2735657.38      6847870.90
#Sta/Elev= 30
  4444.4  455.53  4480.5  455.06  4497.8  453.43  4526.2  452.24  4564.2  451.59
  4577.4  452.21  4600.2  450.10  4652.5  448.43  4663.3  449.01  4668.8  448.82
  4674.5  447.62  4697.2  446.32  4742.9  445.30  4751.8  445.62  4760.2  445.19
  4765.7  444.24  4796.0  442.74  4855.1  442.61  4855.4  442.11  4858.9  442.11
  4859.1  442.61  4981.0  442.79  5087.6  443.37  5096.5  443.33  5103.8  442.70
  5119.2  443.34  5153.3  445.87  5213.4  448.12  5251.5  450.05  5390.2  454.13
#Mann=4,-1,0
  4444.4    0.05       0  4855.1   0.045       0  4859.1    0.05       0
  4981.0   0.045       0
Bank Sta=4855.1,4859.1
Exp/Cntr=0.3,0.1

Type RM Length L Ch R = 1,33687,86,86,86
BEGIN DESCRIPTION:
Mapping XS f282cbba
END DESCRIPTION:
XS GIS Cut Line= 4
      2736373.65      6847399.22      2735974.85      6847585.90
      2735845.63      6847646.48      2735639.46      6847764.09
#Sta/Elev= 30
  4560.9  452.46  4591.4  451.05  4604.2  451.59  4613.5  450.11  4649.9  448.60
  4701.8  448.46  4718.4  446.78  4741.2  445.86  4779.1  445.09  4792.4  445.45
  4809.8  443.38  4843.4  442.32  4843.6  441.82  4847.1  441.82  4847.4  442.32
  4867.5  445.08  4889.5  446.34  4929.4  446.30  4935.0  446.83  4966.8  447.03
  4993.9  446.73  5049.1  447.30  5066.2  447.05  5071.9  446.38  5100.3  446.29
  5132.5  444.40  5140.4  443.37  5189.6  445.93  5280.1  449.40  5381.3  451.68
#Mann=4,-1,0
  4560.9    0.05       0  4843.4   0.045       0  4847.4    0.05       0
  4993.9   0.045       0
Bank Sta=4843.4,4847.4
Exp/Cntr=0.3,0.1

Type RM Length L Ch R = 1,33601,340,340,340
BEGIN DESCRIPTION:
Dry Creek33601
END DESCRIPTION:
XS GIS Cut Line= 3
      2736365.35      6847250.36      2735927.20      6847517.08
      2735620.86      6847682.92
#Sta/Elev= 30
  4492.9  455.42  4506.7  454.91  4522.2  455.29  4537.7  453.43  4559.0  451.95
  4580.3  451.01  4586.2  451.56  4595.8  451.20  4617.1  449.38  4653.9  447.96
  4696.5  447.42  4726.3  445.02  4770.1  444.88  4776.0  444.69  4791.4  442.74
  4878.5  440.93  4886.4  440.02  4929.0  439.35  4965.8  437.94  4981.3  436.60
  5000.6  436.39  5000.8  435.89  5004.3  435.89  5004.6  436.39  5052.7  437.37
  5090.1  441.44  5128.1  442.75  5177.8  445.37  5281.2  448.82  5354.2  450.08
#Mann=3,-1,0
  4492.9    0.05       0  5000.6    0.05       0  5004.6   0.045       0
Bank Sta=5000.6,5004.6
Exp/Cntr=0.3,0.1

Type RM Length L Ch R = 1,33261,296,296,296
BEGIN DESCRIPTION:
Mapping XS e41c643c
END DESCRIPTION:
XS GIS Cut Line= 3
      2736211.37      6846964.50      2735923.61      6847176.32
      2735655.18      6847425.39
#Sta/Elev= 30
  4644.8  451.13  4681.8  449.57  4696.4  448.43  4731.9  447.13  4746.6  446.05
  4752.8  446.20  4782.1  444.60  4817.6  443.60  4832.2  442.50  4932.5  439.44
  4938.7  439.75  4947.1  438.74  4953.3  438.73  4961.8  436.87  4968.0  436.93
  4974.3  435.88  4982.6  435.30  5030.0  434.02  5030.3  433.52  5033.8  433.52
  5034.0  434.02  5053.4  434.06  5067.2  434.82  5074.5  436.09  5081.3  436.38
  5088.7  437.99  5117.0  439.17  5194.7  439.52  5339.4  443.38  5368.3  444.06
#Mann=4,-1,0
  4644.8    0.05       0  5030.0    0.05       0  5034.0    0.05       0
  5339.4   0.045       0
Bank Sta=5030,5034
Exp/Cntr=0.3,0.1

Type RM Length L Ch R = 1,32965,281,281,281
BEGIN DESCRIPTION:
Dry Creek33167.51
END DESCRIPTION:
XS GIS Cut Line= 3
      2736212.70      6846752.39      2735825.60      6846911.17
      2735665.52      6847384.53
#Sta/Elev= 30
  4581.6  452.08  4670.0  447.93  4723.4  446.05  4729.4  445.33  4800.8  442.18
  4830.2  441.67  4854.1  440.20  4923.9  437.47  4931.5  436.15  4936.9  436.23
  4955.5  434.02  4960.9  434.18  4967.1  433.38  4990.3  432.55  4995.1  431.91
  4995.3  431.41  4998.8  431.41  4999.1  431.91  5020.9  433.18  5063.2  432.63
  5072.6  432.76  5074.5  433.26  5077.9  434.16  5104.1  435.79  5115.9  437.84
  5154.4  439.04  5203.7  440.37  5337.6  442.28  5411.5  442.20  5499.7  443.43
#Mann=5,-1,0
  4581.6    0.05       0  4995.1    0.05       0  4999.1    0.05       0
  5074.5   0.045       0  5154.4    0.05       0
Bank Sta=4995.1,4999.1
Exp/Cntr=0.3,0.1

Type RM Length L Ch R = 1,32684,287,287,287
BEGIN DESCRIPTION:
Dry Creek32684.29
END DESCRIPTION:
XS GIS Cut Line= 3
      2736098.85      6846636.49      2735772.47      6846649.54
      2735255.15      6846661.54
#Sta/Elev= 30
  4677.6  446.78  4790.5  441.72  4890.6  437.98  4940.7  436.63  5000.0  432.97
  5004.2  432.97  5010.7  431.96  5028.7  431.31  5028.9  430.81  5032.5  430.81
  5032.8  431.31  5050.7  431.58  5080.7  431.41  5095.8  431.93  5120.7  432.46
  5140.7  435.44  5160.8  435.29  5180.8  434.68  5200.8  435.57  5250.8  436.75
  5279.3  438.04  5284.3  437.72  5300.8  438.40  5320.8  438.66  5370.8  440.41
  5400.8  442.24  5440.8  442.57  5490.8  444.23  5500.8  445.06  5521.7  444.97
#Mann=4,-1,0
  4677.6    0.05       0  5028.7    0.05       0  5032.8    0.05       0
  5095.8   0.045       0
Bank Sta=5028.7,5032.8
Exp/Cntr=0.3,0.1

Type RM Length L Ch R = 1,32397,261,261,261
BEGIN DESCRIPTION:
Dry Creek32396.83
END DESCRIPTION:
XS GIS Cut Line= 3
      2736119.75      6846373.75      2735723.08      6846378.21
      2735276.05      6846398.80
#Sta/Elev= 30
  4606.2  447.10  4620.0  446.78  4660.0  444.98  4700.0  443.99  4820.0  439.81
  4880.0  437.39  4890.0  436.84  4930.0  432.93  4950.0  431.67  4960.0  431.70
  4980.0  430.51  5010.0  431.14  5017.9  430.45  5018.2  429.95  5021.8  429.95
  5022.1  430.45  5050.0  430.80  5060.0  431.71  5070.0  433.12  5080.1  433.65
  5120.1  434.46  5140.1  435.33  5150.1  435.21  5220.2  436.87  5350.3  441.79
  5360.4  442.44  5380.4  442.75  5400.4  443.57  5410.4  443.47  5450.4  444.76
#Mann=3,-1,0
  4606.2    0.05       0  5017.9    0.05       0  5022.1    0.05       0
Bank Sta=5017.9,5022.1
Exp/Cntr=0.3,0.1

Type RM Length L Ch R = 1,32136,308,308,308
BEGIN DESCRIPTION:
Dry Creek32135.95
END DESCRIPTION:
XS GIS Cut Line= 3
      2736167.57      6846114.77      2735726.91      6846117.32
      2735216.09      6846102.63
#Sta/Elev= 30
  4558.4  444.27  4660.0  443.09  4700.0  440.97  4740.0  440.31  4750.0  440.76
  4767.8  439.46  4772.8  440.07  4780.0  439.39  4830.0  438.22  4850.0  436.76
  4860.0  434.76  4870.0  433.79  4900.0  433.31  4950.0  430.48  4960.0  429.67
  4970.0  427.61  4980.0  429.25  4990.0  429.55  4994.9  427.36  4995.2  426.86
  4998.8  426.86  4999.1  427.36  5010.0  428.23  5045.0  433.24  5080.0  433.06
  5210.1  434.79  5330.1  439.20  5389.1  440.55  5470.2  441.36  5510.1  443.22
#Mann=3,-1,0
  4558.4    0.05       0  4994.9    0.05       0  4999.1    0.05       0
Bank Sta=4994.9,4999.1
Exp/Cntr=0.3,0.1

Type RM Length L Ch R = 1,31828,307,307,307
BEGIN DESCRIPTION:
Dry Creek31827.85
END DESCRIPTION:
XS GIS Cut Line= 3
      2736225.78      6845890.15      2735773.49      6845824.89
      2735454.32      6845812.14
#Sta/Elev= 30
  4545.7  441.53  4565.7  441.22  4577.8  441.60  4596.0  440.47  4686.9  438.21
  4707.1  438.75  4727.3  437.22  4838.5  434.61  4929.7  431.83  4949.6  429.80
  4959.7  429.79  4989.9  428.46  4995.0  428.90  4996.7  427.77  4997.0  427.27
  5000.8  427.27  5001.1  427.77  5010.2  428.37  5020.2  428.24  5050.2  430.20
  5070.2  430.83  5080.2  430.53  5100.2  431.32  5120.3  431.34  5180.3  433.91
  5270.4  437.10  5280.4  437.67  5290.4  438.81  5310.4  442.78  5322.1  442.97
#Mann=3,-1,0
  4545.7    0.05       0  4996.7    0.05       0  5001.1    0.05       0
Bank Sta=4996.7,5001.1
Exp/Cntr=0.3,0.1

Type RM Length L Ch R = 1,31521,269,269,269
BEGIN DESCRIPTION:
Dry Creek31520.76
END DESCRIPTION:
XS GIS Cut Line= 3
      2736265.58      6845607.95      2735872.55      6845549.28
      2735331.37      6845515.69
#Sta/Elev= 30
  4606.0  441.78  4635.9  441.11  4646.0  441.54  4666.2  440.02  4716.8  438.40
  4758.5  437.47  4777.5  437.77  4797.7  436.41  4868.5  433.68  4908.9  433.55
  4919.0  433.03  4956.1  428.11  4969.6  427.51  4979.7  425.43  4996.9  425.17
  4997.2  424.67  5001.1  424.67  5001.4  425.17  5003.4  425.17  5009.9  427.30
  5070.1  430.77  5110.1  430.67  5170.3  431.78  5270.4  435.31  5310.5  437.15
  5377.4  438.95  5382.4  438.53  5440.8  439.14  5460.8  439.90  5545.6  441.02
#Mann=3,-1,0
  4606.0    0.05       0  4996.9    0.05       0  5001.4    0.05       0
Bank Sta=4996.9,5001.4
Exp/Cntr=0.3,0.1

Type RM Length L Ch R = 1,31252,174,174,174
BEGIN DESCRIPTION:
Dry Creek31252.38
END DESCRIPTION:
XS GIS Cut Line= 3
      2736386.28      6845345.84      2735970.69      6845312.62
      2735336.35      6845305.40
#Sta/Elev= 30
  4583.0  441.99  4633.4  440.67  4653.5  439.29  4663.5  439.49  4713.7  437.32
  4763.9  436.64  4804.0  434.32  4863.3  432.60  4934.4  431.15  4944.4  430.54
  4953.5  428.96  4958.5  428.91  4984.6  425.37  4992.3  425.36  4992.6  424.86
  4996.5  424.86  4996.8  425.36  5024.6  426.15  5034.6  426.85  5044.6  428.55
  5064.6  429.13  5094.6  428.55  5134.6  428.80  5244.6  431.28  5374.6  437.13
  5434.6  437.07  5504.6  437.80  5580.4  439.87  5621.3  440.40  5634.3  440.58
#Mann=5,-1,0
  4583.0   0.035       0  4863.3   0.063       0  4992.3   0.063       0
  4996.8   0.063       0  5621.3   0.035       0
Bank Sta=4992.3,4996.8
Exp/Cntr=0.3,0.1

Type RM Length L Ch R = 1,31078,270,270,270
BEGIN DESCRIPTION:
Dry Creek31078.25
END DESCRIPTION:
XS GIS Cut Line= 3
      2736404.54      6845135.86      2735990.11      6845144.23
      2735382.19      6845135.03
#Sta/Elev= 30
  4588.4  438.88  4647.0  437.83  4657.0  438.15  4737.0  434.72  4767.0  434.14
  4787.0  434.47  4797.0  433.66  4867.0  432.10  4927.0  429.07  4947.0  427.20
  4967.0  426.66  4987.0  427.19  5002.5  425.40  5024.7  425.13  5025.0  424.63
  5029.0  424.63  5029.3  425.13  5047.0  427.11  5067.0  426.73  5137.0  430.09
  5167.0  429.49  5237.0  430.18  5277.1  431.70  5327.1  432.61  5347.1  434.10
  5367.1  433.43  5427.1  435.92  5497.1  437.72  5544.6  437.91  5610.9  439.95
#Mann=3,-1,0
  4588.4   0.063       0  5024.7   0.063       0  5029.3   0.063       0
Bank Sta=5024.7,5029.3
Exp/Cntr=0.3,0.1

Type RM Length L Ch R = 1,30808,241,241,241
BEGIN DESCRIPTION:
Dry Creek30808.07
END DESCRIPTION:
XS GIS Cut Line= 3
      2736475.64      6844920.73      2736075.13      6844900.85
      2735659.84      6844898.79
#Sta/Elev= 30
  4599.8  437.03  4639.5  436.12  4659.5  436.68  4699.9  434.32  4749.6  434.20
  4759.6  433.28  4819.7  431.03  4900.9  429.92  4909.8  429.58  4919.8  428.52
  4949.9  427.63  4969.9  427.46  4989.9  425.00  5007.6  424.61  5007.9  424.11
  5011.9  424.11  5012.2  424.61  5019.9  424.96  5039.9  424.76  5049.9  425.61
  5059.9  427.43  5069.9  427.88  5099.9  427.35  5139.9  427.51  5159.9  428.63
  5239.9  431.08  5279.9  432.05  5339.9  432.57  5409.9  434.11  5416.1  434.55
#Mann=3,-1,0
  4599.8    0.05       0  5007.6    0.05       0  5012.2    0.05       0
Bank Sta=5007.6,5012.2
Exp/Cntr=0.3,0.1

Type RM Length L Ch R = 1,30567,274,274,274
BEGIN DESCRIPTION:
Dry Creek30566.61
END DESCRIPTION:
XS GIS Cut Line= 3
      2736484.50      6844642.98      2736122.32      6844675.97
      2735821.30      6844733.78
#Sta/Elev= 30
  4639.7  437.57  4658.3  436.28  4688.4  435.31  4728.6  434.99  4738.6  435.37
  4748.6  434.26  4758.7  433.77  4788.8  433.61  4808.9  432.38  4893.9  429.42
  4919.3  427.44  4949.5  426.39  4959.5  426.79  4979.6  421.94  4987.2  421.02
  4987.5  420.52  4991.7  420.52  4992.1  421.02  4999.0  422.70  5050.5  426.63
  5081.1  426.08  5121.8  426.34  5203.3  427.71  5217.1  428.17  5223.6  428.85
  5244.0  429.33  5254.2  430.05  5274.6  433.23  5294.9  434.94  5309.9  434.93
#Mann=3,-1,0
  4639.7    0.05       0  4987.2    0.05       0  4992.1    0.05       0
Bank Sta=4987.2,4992.1
Exp/Cntr=0.3,0.1

Type RM Length L Ch R = 1,30293,293,293,293
BEGIN DESCRIPTION:
Dry Creek30292.98
END DESCRIPTION:
XS GIS Cut Line= 3
      2736253.21      6844446.66      2735921.22      6844508.94
      2735569.76      6844606.76
#Sta/Elev= 30
  4664.3  432.97  4711.1  434.13  4742.9  433.67  4821.3  429.42  4826.4  429.49
  4854.8  427.41  4895.5  425.97  4905.7  424.14  4926.0  423.82  4931.5  423.03
  4956.5  421.90  4966.7  421.86  4976.9  422.49  4984.1  420.31  4986.7  420.08
  4987.0  419.58  4991.2  419.58  4991.6  420.08  4997.1  422.86  5030.9  422.59
  5080.2  425.57  5138.8  426.90  5178.2  427.01  5204.7  428.24  5212.4  429.10
  5217.6  428.72  5235.9  429.37  5251.8  430.58  5325.4  432.70  5366.9  432.90
#Mann=3,-1,0
  4664.3    0.05       0  4986.7    0.05       0  4991.6    0.05       0
Bank Sta=4986.7,4991.6
Exp/Cntr=0.3,0.1

Type RM Length L Ch R = 1,30000,298,298,298
BEGIN DESCRIPTION:
Dry Creek29999.8
END DESCRIPTION:
XS GIS Cut Line= 3
      2736160.90      6844252.25      2735774.75      6844274.28
      2735463.82      6844285.10
#Sta/Elev= 30
  4614.3  433.89  4629.2  433.77  4682.3  432.05  4789.5  427.51  4839.6  426.28
  4879.6  424.40  4899.7  423.95  4909.7  424.38  4919.7  424.15  4929.7  422.77
  4939.7  422.36  4949.7  422.08  4959.8  422.38  4979.8  421.88  4989.8  419.51
  4995.5  418.67  4995.8  418.17  5000.0  418.17  5000.4  418.67  5009.8  421.71
  5019.8  423.62  5052.7  425.79  5079.9  425.70  5149.9  429.17  5169.9  429.75
  5189.9  429.34  5220.0  429.87  5260.0  432.62  5270.0  432.34  5312.2  433.11
#Mann=3,-1,0
  4614.3    0.05       0  4995.5    0.05       0  5000.4    0.05       0
Bank Sta=4995.5,5000.4
Exp/Cntr=0.3,0.1

Type RM Length L Ch R = 1,29702,175,175,175
BEGIN DESCRIPTION:
Dry Creek29702.01
END DESCRIPTION:
XS GIS Cut Line= 3
      2736129.48      6843996.93      2735724.13      6843992.53
      2735375.55      6844010.26
#Sta/Elev= 30
  4596.7  431.99  4640.2  430.37  4683.8  429.62  4860.2  424.15  4910.2  423.25
  4940.2  423.95  4960.2  423.83  4970.2  422.28  4980.2  418.03  4987.7  416.88
  4988.1  416.38  4992.3  416.38  4992.7  416.88  5002.1  417.04  5010.2  419.94
  5020.2  421.09  5030.2  420.72  5040.3  420.81  5060.3  423.95  5090.3  423.97
  5150.4  425.70  5160.4  426.49  5180.4  427.31  5210.5  429.14  5220.5  430.62
  5230.5  431.00  5260.5  431.31  5290.6  433.82  5310.6  433.55  5351.1  433.80
#Mann=3,-1,0
  4596.7    0.05       0  4987.7    0.05       0  4992.7    0.05       0
Bank Sta=4987.7,4992.7
Exp/Cntr=0.3,0.1

Type RM Length L Ch R = 1,29527,322,322,322
BEGIN DESCRIPTION:
Dry Creek29527.3
END DESCRIPTION:
XS GIS Cut Line= 3
      2736150.12      6843807.93      2735754.81      6843828.88
      2735481.28      6843826.73
#Sta/Elev= 30
  4606.8  432.73  4661.0  430.90  4691.0  431.06  4701.0  429.64  4731.1  428.18
  4791.2  427.25  4801.2  425.75  4821.2  424.71  4838.7  416.04  4839.1  415.54
  4843.7  416.04  4851.3  420.28  4881.3  422.09  4891.3  422.30  4901.3  418.81
  4911.3  417.64  4921.4  419.05  4952.3  419.70  4961.4  416.24  4971.4  416.53
  4981.4  420.83  5031.5  422.01  5041.5  424.01  5081.5  423.20  5171.5  424.75
  5191.5  425.83  5211.5  428.01  5231.5  428.47  5251.5  430.76  5276.2  430.83
#Mann=3,-1,0
  4606.8    0.05       0  4838.7    0.05       0  4843.7    0.05       0
Bank Sta=4838.7,4843.7
Exp/Cntr=0.3,0.1

Type RM Length L Ch R = 1,29205,461,461,461
BEGIN DESCRIPTION:
Dry Creek29205.14
END DESCRIPTION:
XS GIS Cut Line= 3
      2736168.51      6843574.57      2735921.94      6843594.72
      2735546.92      6843611.82
#Sta/Elev= 30
  4757.4  430.69  4790.0  429.72  4850.2  427.00  4880.3  426.34  4910.4  424.29
  4960.6  422.92  4990.7  415.26  5004.8  415.16  5008.2  413.99  5008.6  413.49
  5012.9  413.49  5013.2  413.99  5020.8  419.10  5029.4  421.08  5060.8  421.81
  5090.8  419.52  5110.8  420.42  5120.9  420.04  5140.9  421.85  5150.9  422.11
  5170.9  421.94  5190.9  422.37  5231.0  421.70  5254.2  423.62  5291.0  423.38
  5331.1  425.12  5351.1  427.19  5361.1  429.77  5377.0  435.28  5380.2  435.62
#Mann=4,-1,0
  4757.4    0.05       0  5008.2    0.05       0  5013.2    0.05       0
  5377.0   0.033       0
Bank Sta=5008.2,5013.2
Exp/Cntr=0.3,0.1

Type RM Length L Ch R = 1,28744,384,384,384
BEGIN DESCRIPTION:
Dry Creek28613.66
END DESCRIPTION:
XS GIS Cut Line= 3
      2736218.74      6843169.86      2735776.44      6843206.27
      2735325.02      6843229.22
#Sta/Elev= 30
  4556.2  436.36  4599.1  433.61  4619.2  434.28  4639.2  431.64  4669.3  429.79
  4739.6  428.64  4769.7  425.85  4819.8  424.84  4839.9  425.43  4860.0  422.73
  4900.1  420.16  4960.3  420.28  4970.3  417.82  4980.4  413.17  4987.8  412.75
  4988.2  412.25  4993.0  412.75  4996.0  418.71  5010.5  419.45  5030.5  418.67
  5060.5  420.61  5100.6  419.86  5180.7  420.83  5220.7  422.97  5230.7  424.20
  5260.8  424.22  5290.8  427.15  5340.9  428.13  5387.2  431.90  5452.0  432.19
#Mann=3,-1,0
  4556.2    0.05       0  4987.8    0.05       0  4993.0    0.05       0
Bank Sta=4987.8,4993
Exp/Cntr=0.3,0.1

Type RM Length L Ch R = 1,28360,382,382,382
BEGIN DESCRIPTION:
Dry Creek28360.3
END DESCRIPTION:
XS GIS Cut Line= 3
      2736040.72      6842843.12      2735682.35      6842856.28
      2735303.04      6842901.42
#Sta/Elev= 30
  4642.3  430.99  4677.0  430.21  4687.1  430.79  4716.4  427.48  4721.4  427.74
  4727.1  426.91  4747.1  426.16  4767.1  426.86  4787.1  424.12  4827.1  421.64
  4867.2  420.45  4897.2  418.37  4907.2  419.12  4947.2  416.31  4987.3  418.53
  5000.9  418.45  5017.4  416.80  5024.8  411.34  5025.3  410.84  5029.7  410.84
  5030.1  411.34  5037.5  411.68  5047.6  417.20  5067.7  418.29  5148.3  418.34
  5228.9  420.91  5259.1  424.64  5289.3  425.10  5319.5  428.21  5382.9  429.67
#Mann=3,-1,0
  4642.3    0.05       0  5024.8    0.05       0  5030.1    0.05       0
Bank Sta=5024.8,5030.1
Exp/Cntr=0.3,0.1

Type RM Length L Ch R = 1,27978,246,246,246
BEGIN DESCRIPTION:
Dry Creek27977.86
END DESCRIPTION:
XS GIS Cut Line= 3
      2736049.78      6842538.11      2735573.39      6842572.29
      2735274.69      6842623.67
#Sta/Elev= 30
  4525.7  431.35  4539.5  431.50  4559.6  429.19  4589.6  427.18  4640.4  426.24
  4649.8  424.62  4689.9  421.68  4730.0  420.65  4770.1  418.41  4790.2  418.74
  4800.2  417.80  4860.3  416.86  4920.5  417.96  4969.1  416.54  4980.6  414.31
  4990.7  410.77  4996.8  409.54  4997.2  409.04  5001.7  409.04  5002.1  409.54
  5003.3  409.54  5010.8  417.23  5031.1  416.60  5071.7  421.11  5080.5  421.38
  5087.6  420.74  5132.6  423.14  5152.9  425.28  5201.7  424.58  5306.4  425.50
#Mann=6,-1,0
  4525.7    0.05       0  4969.1    0.12       0  4996.8    0.07       0
  5002.1    0.12       0  5087.6    0.16       0  5201.7    0.05       0
Bank Sta=4996.8,5002.1
Exp/Cntr=0.3,0.1

Type RM Length L Ch R = 1,27732,211,211,211
BEGIN DESCRIPTION:
Dry Creek27732.15
END DESCRIPTION:
XS GIS Cut Line= 3
      2735992.14      6842179.58      2735524.16      6842402.27
      2735234.36      6842544.77
#Sta/Elev= 30
  4486.6  429.86  4515.5  429.15  4523.0  427.55  4545.7  425.39  4568.4  424.69
  4582.0  425.34  4613.8  421.45  4648.4  421.50  4670.6  418.71  4726.0  417.05
  4920.1  415.81  4936.4  416.20  4944.7  417.33  4988.2  416.65  5001.1  413.84
  5004.9  413.84  5008.2  409.99  5008.6  409.49  5013.1  409.49  5013.5  409.99
  5016.4  410.48  5025.1  415.08  5033.3  416.46  5083.8  419.82  5123.2  420.62
  5128.8  421.40  5158.8  421.39  5200.8  423.33  5218.7  424.13  5327.8  425.19
#Mann=5,-1,0
  4486.6    0.05       0  4944.7    0.12       0  5008.2    0.07       0
  5013.5    0.12       0  5200.8    0.16       0
Bank Sta=5008.2,5013.5
Exp/Cntr=0.3,0.1

Type RM Length L Ch R = 1,27521,401,401,401
BEGIN DESCRIPTION:
Dry Creek27521.11
END DESCRIPTION:
XS GIS Cut Line= 3
      2735879.79      6842038.38      2735427.42      6842222.48
      2735076.61      6842380.87
#Sta/Elev= 30
  4519.4  428.60  4534.3  428.36  4545.1  426.56  4569.1  424.57  4609.9  424.55
  4641.3  420.77  4653.0  420.26  4670.8  420.96  4700.2  417.51  4717.8  417.69
  4729.7  416.45  4761.0  415.73  4894.4  415.92  4944.5  416.52  4955.3  414.35
  4962.4  409.06  4965.1  408.91  4965.6  408.41  4970.1  408.41  4970.5  408.91
  4976.9  410.44  4986.5  416.54  5031.3  415.82  5044.2  417.11  5097.1  417.59
  5154.7  420.10  5234.7  423.22  5257.8  422.78  5289.2  423.26  5392.7  425.84
#Mann=6,-1,0
  4519.4    0.05       0  4894.4    0.12       0  4965.1    0.07       0
  4970.5    0.12       0  5154.7    0.16       0  5289.2    0.05       0
Bank Sta=4965.1,4970.5
Exp/Cntr=0.3,0.1

Type RM Length L Ch R = 1,27120,309,309,309
BEGIN DESCRIPTION:
Dry Creek27120.31
END DESCRIPTION:
XS GIS Cut Line= 3
      2735655.01      6841786.54      2735324.88      6841955.38
      2734936.09      6842182.57
#Sta/Elev= 30
  4632.0  428.49  4678.1  427.20  4700.3  427.64  4716.9  426.00  4722.5  424.49
  4805.7  420.26  4833.6  416.99  4884.2  414.98  4911.2  414.66  4922.9  413.12
  4929.4  413.63  4939.0  415.02  4961.2  414.93  4967.8  413.28  4977.8  414.07
  4983.4  409.12  4999.4  412.47  5002.8  412.47  5005.7  408.20  5018.7  407.48
  5019.1  406.98  5024.1  407.48  5036.2  413.56  5042.8  414.48  5132.3  416.33
  5256.1  417.73  5296.2  419.22  5400.8  423.10  5416.5  425.45  5453.1  427.68
#Mann=7,-1,0
  4632.0    0.05       0  4884.2    0.12       0  4929.4    0.16       0
  5018.7    0.07       0  5024.1    0.16       0  5132.3    0.12       0
  5296.2    0.05       0
Bank Sta=5018.7,5024.1
Exp/Cntr=0.3,0.1

Type RM Length L Ch R = 1,26811,266,266,266
BEGIN DESCRIPTION:
Dry Creek26810.78
END DESCRIPTION:
XS GIS Cut Line= 3
      2735571.83      6841576.76      2735222.07      6841737.34
      2734829.30      6841927.17
#Sta/Elev= 30
  4618.9  427.21  4669.9  426.51  4692.9  427.52  4746.4  423.81  4790.4  422.48
  4801.4  422.91  4830.8  419.20  4877.7  417.12  4928.3  414.49  4951.3  414.01
  4979.8  412.09  4985.7  407.67  4986.1  407.17  4991.1  407.67  4997.2  408.67
  5002.2  411.18  5025.4  415.20  5048.0  413.61  5098.7  413.75  5206.2  415.42
  5243.7  418.70  5266.0  418.92  5321.3  421.50  5332.6  421.70  5387.0  425.38
  5409.6  426.36  5415.1  425.90  5421.4  427.09  5433.3  427.82  5440.0  428.61
#Mann=7,-1,0
  4618.9    0.05       0  4877.7    0.16       0  4985.7    0.07       0
  4991.1    0.16       0  5098.7    0.12       0  5321.3    0.16       0
  5433.3    0.05       0
Bank Sta=4985.7,4991.1
Exp/Cntr=0.3,0.1

Type RM Length L Ch R = 1,26545,324,324,324
BEGIN DESCRIPTION:
Dry Creek26544.83
END DESCRIPTION:
XS GIS Cut Line= 3
      2735471.14      6841361.38      2735183.06      6841523.40
      2734765.36      6841762.89
#Sta/Elev= 30
  4674.2  426.30  4728.1  424.38  4781.6  420.11  4817.8  418.77  4846.6  415.92
  4868.3  416.05  4874.8  415.23  4927.6  412.91  4933.3  413.51  4970.9  413.33
  4978.4  412.53  5030.1  412.98  5035.9  411.86  5045.9  407.33  5049.0  405.11
  5049.4  404.61  5054.4  405.11  5067.5  413.97  5073.3  414.40  5082.0  413.25
  5104.9  412.79  5169.6  413.43  5283.4  417.72  5352.3  420.95  5395.5  425.18
  5425.8  426.39  5439.4  427.76  5470.3  428.30  5476.0  429.21  5486.2  428.82
#Mann=6,-1,0
  4674.2    0.05       0  4874.8    0.12       0  5049.0    0.07       0
  5054.4    0.12       0  5283.4    0.16       0  5425.8    0.05       0
Bank Sta=5049,5054.4
Exp/Cntr=0.3,0.1

Type RM Length L Ch R = 1,26221,416,416,416
BEGIN DESCRIPTION:
Dry Creek26221.24
END DESCRIPTION:
XS GIS Cut Line= 3
      2735352.93      6841142.96      2735122.88      6841272.60
      2734750.34      6841491.99
#Sta/Elev= 30
  4739.7  425.86  4793.6  424.65  4830.6  422.85  4933.1  415.85  4949.0  414.13
  4962.9  413.68  4974.0  413.16  4992.4  411.91  4996.3  404.30  4996.8  403.80
  5001.4  403.80  5001.8  404.30  5014.0  406.09  5023.4  411.96  5029.7  412.85
  5035.5  413.04  5058.2  411.38  5071.1  411.58  5081.4  412.54  5103.9  411.72
  5168.3  412.60  5183.9  413.91  5205.4  413.98  5242.5  415.33  5324.5  419.09
  5371.5  421.40  5386.9  422.36  5402.6  424.15  5429.8  425.14  5436.1  425.81
#Mann=7,-1,0
  4739.7    0.05       0  4962.9    0.16       0  4974.0    0.12       0
  4996.3    0.07       0  5001.8    0.12       0  5071.1    0.16       0
  5324.5    0.05       0
Bank Sta=4996.3,5001.8
Exp/Cntr=0.3,0.1

Type RM Length L Ch R = 1,25805,324,324,324
BEGIN DESCRIPTION:
Dry Creek25805.31
END DESCRIPTION:
XS GIS Cut Line= 3
      2735309.49      6840975.90      2734920.10      6840979.68
      2734664.81      6840980.14
#Sta/Elev= 30
  4615.7  424.45  4649.2  423.82  4709.2  419.78  4759.2  415.22  4809.4  412.55
  4839.2  411.27  4879.2  411.76  4889.2  410.88  4899.2  410.73  4919.2  411.58
  4929.2  411.01  4949.2  410.80  4979.2  411.01  4989.2  404.68  4996.5  403.14
  4996.9  402.64  5001.5  402.64  5002.0  403.14  5004.7  405.14  5009.7  405.14
  5019.2  410.79  5029.2  411.77  5049.2  412.96  5099.2  414.93  5129.2  417.08
  5149.2  419.01  5199.2  422.39  5219.2  423.13  5229.2  423.95  5260.4  424.72
#Mann=4,-1,0
  4615.7    0.05       0  4809.4    0.12       0  4996.5    0.07       0
  5002.0    0.12       0
Bank Sta=4996.5,5002
Exp/Cntr=0.3,0.1

Type RM Length L Ch R = 1,25481,226,226,226
BEGIN DESCRIPTION:
Dry Creek25480.541
END DESCRIPTION:
XS GIS Cut Line= 3
      2735353.93      6840784.73      2734875.46      6840724.82
      2734652.98      6840700.61
#Sta/Elev= 30
  4517.8  422.24  4556.0  419.80  4584.6  417.09  4589.7  417.57  4626.6  415.15
  4707.2  411.93  4787.8  409.90  4826.3  410.14  4848.3  409.42  4870.7  409.66
  4878.5  410.05  4949.1  410.59  4959.1  409.55  4966.5  402.23  4966.9  401.73
  4971.5  401.73  4972.0  402.23  4979.3  402.75  4987.4  406.69  4992.5  410.80
  4997.2  411.60  5019.6  412.77  5059.8  417.04  5083.3  418.65  5090.0  419.77
  5120.2  421.77  5140.3  422.59  5169.7  422.74  5190.6  423.49  5223.8  423.45
#Mann=4,-1,0
  4517.8    0.05       0  4870.7    0.12       0  4966.5    0.07       0
  4972.0    0.12       0
Bank Sta=4966.5,4972
Exp/Cntr=0.3,0.1

Type RM Length L Ch R = 1,25255,455,455,455
BEGIN DESCRIPTION:
Dry Creek25254.88
END DESCRIPTION:
XS GIS Cut Line= 3
      2735264.78      6840661.06      2734926.63      6840515.37
      2734240.33      6840307.12
#Sta/Elev= 30
  4631.6  414.84  4750.5  409.48  4920.6  409.38  4951.1  407.78  4956.9  406.22
  4989.6  410.30  4999.0  404.32  5002.7  404.32  5008.2  401.09  5008.6  400.59
  5013.7  401.09  5021.4  409.67  5067.4  410.23  5084.1  413.07  5133.2  416.35
  5237.1  417.61  5349.7  412.20  5387.1  410.71  5439.4  410.89  5445.0  406.88
  5450.2  406.32  5460.3  410.46  5469.8  410.68  5516.0  411.61  5543.7  412.92
  5554.3  414.74  5572.5  414.66  5581.8  414.02  5675.1  420.34  5717.0  423.53
#Mann=8,-1,0
  4631.6    0.05       0  4951.1    0.12       0  5008.2    0.07       0
  5013.7    0.12       0  5349.7    0.16       0  5469.8   0.035       0
  5572.5    0.07       0  5675.1    0.05       0
Bank Sta=5008.2,5013.7
Exp/Cntr=0.3,0.1

Type RM Length L Ch R = 1,24800,261,261,261
BEGIN DESCRIPTION:
Dry Creek24799.52
END DESCRIPTION:
XS GIS Cut Line= 3
      2735817.16      6840131.20      2734748.38      6840131.90
      2734249.70      6840120.11
#Sta/Elev= 30
  3930.0  423.75  3991.2  419.47  4031.2  420.90  4055.9  418.04  4111.2  413.73
  4166.6  411.31  4371.2  407.87  4391.2  408.64  4441.2  406.08  4451.2  408.25
  4471.2  407.85  4511.2  409.51  4781.2  407.17  4967.4  408.21  5011.2  408.79
  5018.1  401.31  5018.6  400.81  5024.3  401.31  5031.2  401.52  5041.2  407.77
  5066.4  408.20  5141.2  409.12  5151.2  408.03  5161.2  402.65  5171.2  409.61
  5264.3  411.07  5311.2  411.84  5331.3  415.70  5363.2  417.85  5497.6  423.82
#Mann=9,-1,0
  3930.0    0.05       0  4055.9    0.07       0  4166.6    0.05       0
  4967.4    0.12       0  5018.1    0.07       0  5024.3    0.12       0
  5066.4    0.16       0  5264.3   0.063       0  5363.2    0.05       0
Bank Sta=5018.1,5024.3
Exp/Cntr=0.3,0.1

Type RM Length L Ch R = 1,24539,647,647,647
BEGIN DESCRIPTION:
Dry Creek24539.21
END DESCRIPTION:
XS GIS Cut Line= 3
      2735666.84      6839963.99      2734625.00      6839944.54
      2734220.33      6839934.98
#Sta/Elev= 30
  3958.9  422.69  4069.8  412.66  4119.8  410.05  4209.8  408.80  4229.8  410.77
  4239.8  410.44  4249.8  407.98  4289.8  407.08  4299.8  405.16  4309.8  406.43
  4329.8  405.23  4386.0  408.07  4445.9  408.43  4659.9  406.06  4699.9  407.45
  4969.9  407.76  4979.9  406.78  4989.9  400.23  4994.8  400.20  4995.3  399.70
  5001.0  400.20  5002.9  400.20  5009.9  408.31  5039.7  408.12  5069.9  406.54
  5099.9  409.92  5138.6  408.03  5233.9  412.16  5320.0  417.05  5405.7  419.81
#Mann=7,-1,0
  3958.9    0.05       0  4445.9    0.12       0  4994.8    0.07       0
  5001.0    0.12       0  5039.7   0.063       0  5138.6    0.16       0
  5233.9    0.05       0
Bank Sta=4994.8,5001
Exp/Cntr=0.3,0.1

Type RM Length L Ch R = 1,23892,181,181,181
BEGIN DESCRIPTION:
Dry Creek23891.61
END DESCRIPTION:
XS GIS Cut Line= 5
      2734719.78      6838974.04      2734709.55      6839406.73
      2734666.55      6839610.07      2734599.82      6839698.54
      2734154.38      6839906.12
#Sta/Elev= 30
  4580.0  417.05  4797.0  418.72  4894.5  415.05  4907.1  414.92  4917.1  412.99
  4951.8  410.71  4957.1  408.20  4967.1  405.22  4977.1  404.45  4991.5  398.52
  4992.0  398.02  5002.6  398.52  5012.4  400.73  5017.5  400.73  5027.4  402.63
  5053.6  403.71  5058.7  405.97  5075.5  406.51  5278.9  405.93  5285.2  407.77
  5293.5  407.09  5299.8  409.24  5340.1  408.97  5350.7  408.92  5368.0  406.23
  5527.4  406.80  5607.8  409.72  5653.5  411.94  5688.7  414.70  5822.9  420.86
#Mann=7,-1,0
  4580.0    0.05       0  4894.5    0.16       0  4991.5    0.07       0
  5002.6    0.16       0  5075.5   0.035       0  5340.1    0.16       0
  5527.4    0.05       0
Bank Sta=4991.5,5002.6
Exp/Cntr=0.3,0.1

Type RM Length L Ch R = 1,23711,296,296,296
BEGIN DESCRIPTION:
Dry Creek23711.14
END DESCRIPTION:
XS GIS Cut Line= 6
      2734563.89      6838980.72      2734548.87      6839243.61
      2734539.88      6839375.01      2734504.23      6839516.18
      2734393.04      6839620.92      2734112.76      6839794.39
#Sta/Elev= 30
  4619.4  411.83  4667.4  412.55  4672.4  412.21  4749.9  414.28  4820.0  414.11
  4840.0  413.55  4850.2  412.15  4910.2  408.98  4918.9  407.81  4940.2  406.02
  4960.3  405.56  4970.3  404.69  4980.3  401.23  4990.4  399.20  4991.2  398.32
  4991.7  397.82  5001.8  397.82  5002.3  398.32  5009.9  401.18  5014.4  401.18
  5020.6  404.70  5030.9  405.56  5144.4  404.82  5260.2  405.21  5312.8  405.36
  5340.1  406.15  5398.0  406.78  5485.7  408.89  5592.9  416.66  5642.4  418.64
#Mann=5,-1,0
  4619.4    0.07       0  4918.9    0.16       0  4991.2    0.07       0
  5002.3    0.16       0  5260.2    0.05       0
Bank Sta=4991.2,5002.3
Exp/Cntr=0.3,0.1

Type RM Length L Ch R = 1,23415,589,589,589
BEGIN DESCRIPTION:
Dry Creek23415.43
END DESCRIPTION:
XS GIS Cut Line= 3
      2734655.15      6838768.99      2734388.85      6839126.40
      2734060.20      6839730.25
#Sta/Elev= 30
  4556.2  414.71  4593.2  414.20  4599.5  412.73  4626.9  411.94  4634.9  410.87
  4649.5  410.58  4798.1  408.67  4828.9  409.35  4849.7  408.29  4864.3  408.83
  4929.0  407.44  4949.8  405.79  4970.7  405.53  4979.0  405.00  4994.3  397.66
  4994.8  397.16  5005.4  397.66  5015.6  401.80  5037.4  404.62  5075.4  403.68
  5118.6  404.43  5259.4  404.27  5382.9  405.99  5473.4  408.83  5598.8  414.69
  5626.3  417.17  5648.1  418.59  5664.3  418.59  5670.0  419.80  5689.4  420.72
#Mann=7,-1,0
  4556.2   0.063       0  4626.9    0.07       0  4798.1   0.035       0
  4994.3   0.035       0  5005.4   0.035       0  5118.6    0.16       0
  5259.4    0.05       0
Bank Sta=4994.3,5005.4
Exp/Cntr=0.3,0.1

Type RM Length L Ch R = 1,22826,248,248,248
BEGIN DESCRIPTION:
Dry Creek22826.07
END DESCRIPTION:
XS GIS Cut Line= 3
      2734664.19      6838706.47      2734173.79      6838710.03
      2733726.95      6838734.12
#Sta/Elev= 30
  4511.9  414.53  4530.1  414.36  4540.1  413.53  4560.4  410.60  4570.1  409.13
  4610.1  407.77  4630.1  406.05  4659.4  404.76  4750.1  403.21  4939.1  403.56
  4950.1  403.84  4960.1  401.54  4964.4  395.20  4964.9  394.70  4975.4  394.70
  4975.9  395.20  4980.1  395.63  4990.1  400.05  5011.9  402.14  5030.1  403.44
  5070.2  402.79  5154.8  403.03  5220.4  404.30  5280.5  407.00  5297.2  408.72
  5310.5  409.14  5353.3  412.63  5380.7  414.88  5410.7  416.54  5449.8  417.44
#Mann=9,-1,0
  4511.9   0.063       0  4560.4    0.07       0  4659.4   0.035       0
  4939.1    0.07       0  4964.4    0.07       0  4975.9    0.07       0
  5011.9   0.035       0  5154.8    0.05       0  5353.3    0.16       0
Bank Sta=4964.4,4975.9
Exp/Cntr=0.3,0.1

Type RM Length L Ch R = 1,22578,313,313,313
BEGIN DESCRIPTION:
Dry Creek22578.19
END DESCRIPTION:
XS GIS Cut Line= 3
      2734638.78      6838461.25      2734070.40      6838499.78
      2733665.00      6838479.38
#Sta/Elev= 30
  4436.8  411.57  4449.6  411.62  4459.6  411.11  4505.9  407.96  4519.8  407.76
  4559.9  405.18  4650.0  402.21  4700.2  401.55  4830.5  402.62  4880.6  402.30
  4948.2  402.72  4960.8  403.16  4970.8  401.77  4980.8  399.24  4990.9  399.05
  5000.4  395.39  5000.9  394.89  5011.4  394.89  5011.9  395.39  5040.9  402.22
  5061.0  401.54  5083.8  401.48  5111.0  402.10  5131.0  403.20  5188.1  404.57
  5271.2  406.21  5301.3  407.85  5341.3  410.78  5371.3  411.89  5412.4  414.54
#Mann=4,-1,0
  4436.8   0.035       0  5000.4   0.035       0  5011.9   0.035       0
  5188.1    0.16       0
Bank Sta=5000.4,5011.9
Exp/Cntr=0.3,0.1

Type RM Length L Ch R = 1,22265,296,296,296
BEGIN DESCRIPTION:
Dry Creek22264.62
END DESCRIPTION:
XS GIS Cut Line= 3
      2734804.79      6838198.91      2734077.10      6838216.36
      2733610.72      6838226.98
#Sta/Elev= 30
  4279.9  408.71  4358.0  407.56  4398.7  406.93  4408.7  407.95  4428.7  407.90
  4438.7  407.20  4448.7  404.23  4458.7  404.63  4588.8  400.54  4768.8  400.20
  4858.9  401.29  4938.9  401.11  4958.9  401.85  4968.9  400.78  4978.9  397.08
  4982.6  394.35  4983.1  393.85  4993.6  393.85  4994.1  394.35  4998.9  401.34
  5005.9  402.12  5168.9  400.08  5204.3  401.24  5249.0  403.46  5269.0  406.14
  5309.0  410.00  5349.0  412.97  5369.0  412.75  5411.4  413.95  5474.3  413.95
#Mann=6,-1,0
  4279.9    0.05       0  4358.0   0.035       0  4982.6   0.035       0
  4994.1   0.035       0  5204.3    0.16       0  5411.4    0.05       0
Bank Sta=4982.6,4994.1
Exp/Cntr=0.3,0.1

Type RM Length L Ch R = 1,21969,436,436,436
BEGIN DESCRIPTION:
Dry Creek21968.73
END DESCRIPTION:
XS GIS Cut Line= 3
      2734853.97      6837827.74      2734116.78      6837935.88
      2733484.27      6838124.42
#Sta/Elev= 30
  4264.5  412.81  4319.7  407.76  4384.5  404.78  4424.2  404.02  4459.4  405.24
  4474.7  402.43  4524.2  401.15  4707.2  399.37  4822.4  399.69  4835.9  399.81
  4899.2  400.69  4929.5  399.80  4982.0  400.76  4990.2  399.84  5000.3  394.56
  5007.1  393.85  5007.6  393.35  5018.6  393.85  5020.8  400.31  5031.3  401.17
  5079.1  399.70  5218.3  399.51  5255.3  399.56  5293.7  402.55  5314.6  405.80
  5326.9  406.88  5411.2  407.62  5536.2  409.54  5607.8  409.61  5669.6  408.11
#Mann=10,-1,0
  4264.5    0.05       0  4384.5   0.035       0  4822.4    0.05       0
  4835.9   0.035       0  4982.0    0.07       0  5007.1    0.07       0
  5018.6    0.07       0  5218.3    0.16       0  5314.6    0.07       0
  5411.2    0.05       0
Bank Sta=5007.1,5018.6
Exp/Cntr=0.3,0.1

Type RM Length L Ch R = 1,21533,346,346,346
BEGIN DESCRIPTION:
Dry Creek21532.55
END DESCRIPTION:
XS GIS Cut Line= 3
      2734540.00      6836811.59      2733870.53      6837631.33
      2733470.68      6838089.12
#Sta/Elev= 30
  3959.5  415.75  4011.1  411.24  4182.0  402.72  4281.5  399.88  4395.9  398.14
  4622.8  397.30  4744.1  398.54  4849.6  398.37  4914.2  399.98  4942.3  398.70
  4950.2  400.01  4979.2  400.36  4985.3  400.31  4991.8  395.90  4999.7  396.44
  5000.4  393.09  5000.9  392.59  5012.0  393.09  5014.1  393.23  5017.5  395.61
  5021.0  395.61  5034.9  400.32  5112.7  398.41  5219.0  399.07  5299.0  398.20
  5368.0  399.06  5389.2  400.87  5431.6  401.10  5517.1  404.89  5625.7  407.69
#Mann=5,-1,0
  3959.5    0.05       0  4979.2    0.07       0  5000.4    0.07       0
  5012.0    0.07       0  5299.0    0.05       0
Bank Sta=5000.4,5012
Exp/Cntr=0.3,0.1

Type RM Length L Ch R = 1,21187,1105,1105,1105
BEGIN DESCRIPTION:
Dry Creek21187.01
END DESCRIPTION:
XS GIS Cut Line= 3
      2733994.09      6836443.61      2733640.39      6837422.41
      2733401.19      6838066.06
#Sta/Elev= 30
  3971.2  416.58  3975.5  416.62  4056.9  410.97  4069.0  410.88  4106.6  407.20
  4130.3  407.22  4138.5  405.58  4160.1  403.79  4273.0  397.97  4404.4  395.98
  4421.0  394.42  4426.3  395.69  4436.3  396.11  4809.0  397.67  4957.3  399.38
  4967.9  399.04  4977.0  391.44  4982.3  392.80  4983.4  391.14  4983.9  390.64
  4995.0  391.14  4999.8  392.58  5007.6  397.29  5011.0  394.61  5021.1  398.29
  5031.8  399.22  5129.1  397.63  5436.3  398.11  5527.4  401.49  5698.6  405.67
#Mann=6,-1,0
  3971.2    0.05       0  3975.5    0.16       0  4056.9    0.12       0
  4160.1    0.05       0  4983.4    0.05       0  4995.0    0.05       0
Bank Sta=4983.4,4995
Exp/Cntr=0.3,0.1

Type RM Length L Ch R = 1,20082,409,409,409
BEGIN DESCRIPTION:
Dry Creek20082.27
END DESCRIPTION:
XS GIS Cut Line= 3
      2733312.57      6836527.17      2733297.16      6836868.80
      2733270.76      6837987.71
#Sta/Elev= 30
  4666.0  417.84  4679.8  417.93  4697.9  416.02  4702.9  416.60  4800.0  409.11
  4870.0  402.44  4924.0  399.51  4930.1  397.84  4970.1  395.35  4974.2  389.75
  4974.7  389.25  4986.2  389.75  4990.2  390.44  5000.2  396.07  5039.1  396.70
  5060.2  395.59  5100.2  395.37  5367.6  396.89  5410.3  396.83  5420.3  397.36
  5440.3  400.79  5450.3  400.99  5470.3  399.52  5490.3  396.56  5537.5  396.44
  5620.4  396.27  5910.4  398.66  5980.5  400.37  6050.5  400.86  6127.2  403.74
#Mann=6,-1,0
  4666.0    0.12       0  4974.2    0.07       0  4986.2    0.12       0
  5039.1    0.05       0  5367.6    0.16       0  5537.5    0.05       0
Bank Sta=4974.2,4986.2
Exp/Cntr=0.3,0.1

Type RM Length L Ch R = 1,19673,350,350,350
BEGIN DESCRIPTION:
Dry Creek19673.34
END DESCRIPTION:
XS GIS Cut Line= 3
      2733051.21      6836551.28      2733027.85      6837074.59
      2733001.72      6837870.63
#Sta/Elev= 30
  4489.6  414.74  4659.5  413.03  4709.5  411.89  4716.5  410.50  4799.6  403.37
  4829.7  398.98  4839.7  398.19  4849.7  395.72  4869.7  395.85  4899.7  394.43
  4943.7  395.82  4959.8  394.83  4969.8  388.64  4973.8  388.03  4974.3  387.53
  4985.3  387.53  4985.8  388.03  4989.8  392.89  4999.8  395.66  5028.2  395.06
  5069.9  394.45  5179.9  395.55  5250.0  394.77  5510.1  396.41  5590.1  398.75
  5620.2  400.01  5630.2  401.14  5650.2  401.43  5754.4  406.58  5809.9  407.78
#Mann=5,-1,0
  4489.6    0.12       0  4973.8    0.07       0  4985.8    0.12       0
  5028.2    0.05       0  5754.4    0.07       0
Bank Sta=4973.8,4985.8
Exp/Cntr=0.3,0.1

Type RM Length L Ch R = 1,19323,275,275,275
BEGIN DESCRIPTION:
Dry Creek19323.22
END DESCRIPTION:
XS GIS Cut Line= 3
      2732968.73      6836471.53      2732781.75      6836924.28
      2732480.67      6837742.40
#Sta/Elev= 30
  4524.4  413.45  4597.3  411.36  4619.5  410.63  4624.9  409.42  4696.7  408.27
  4702.1  407.36  4718.6  408.48  4750.7  406.75  4767.9  405.76  4856.4  399.16
  4885.7  396.01  4939.0  394.40  4992.2  394.74  4993.9  387.58  4994.4  387.08
  5005.9  387.58  5009.8  389.38  5014.2  389.38  5016.2  393.51  5032.1  394.67
  5128.4  394.03  5279.7  393.69  5446.5  395.12  5512.8  396.32  5615.0  400.78
  5660.7  402.99  5671.4  401.97  5703.4  403.94  5765.6  405.63  5886.0  411.50
#Mann=8,-1,0
  4524.4    0.12       0  4597.3    0.16       0  4750.7    0.05       0
  4767.9    0.16       0  4993.9    0.07       0  5005.9    0.16       0
  5128.4    0.05       0  5615.0    0.16       0
Bank Sta=4993.9,5005.9
Exp/Cntr=0.3,0.1
