--- Dry Lacy Fork.prj (project) ---

Proj Title=Dry Lacy Fork Base Level Engineering
Current Plan=p01
Default Exp/Contr=0.3,0.1
English Units
Geom File=g01
Flow File=f01
Plan File=p01
BEGIN DESCRIPTION:
Dry Lacy Fork
END DESCRIPTION:

--- Dry Lacy Fork.p01 (plan) ---

Plan Title=Multiple Run
Short Identifier=Multiple
Geom File=g01
Flow File=f01
Subcritical Flow
K Sum by GR= 0
Std Step Tol= 0.01
Critical Tol= 0.01
Num of Std Step Trials= 20
Max Error Tol= 0.3
Flow Tol Ratio= 0.001
Split Flow NTrial= 30
Split Flow Tol= 0.02
Split Flow Ratio= 0.02
Log Output Level= 0
Friction Slope Method= 1
Unsteady Friction Slope Method= 2
Unsteady Bridges Friction Slope Method= 1
Parabolic Critical Depth
Global Vel Dist=  1 , 1 , 1
Global Log Level= 0
CheckData=True
Encroach Param= -1, 0, 0, 0
BEGIN DESCRIPTION:
Multiple Run
END DESCRIPTION:

--- Dry Lacy Fork.f01 (steady flow) ---

Flow Title=Multiple
Number of Profiles=7
Profile Names=10-year,25-year,50-year,1pct_min,100-year,1pct_plu,500-year
River Rch & RM= Dry Lacy Fork,Reach-1,58313
     132     159     180     101     202     404     255
River Rch & RM= Dry Lacy Fork,Reach-1,56986
     243     309     359     208     415     828     556
River Rch & RM= Dry Lacy Fork,Reach-1,54813
     435     572     683     405     808    1612    1134
River Rch & RM= Dry Lacy Fork,Reach-1,52667
     530     707     849     508    1013    2021    1442
River Rch & RM= Dry Lacy Fork,Reach-1,52028
     620     831    1003     602    1201    2395    1722
River Rch & RM= Dry Lacy Fork,Reach-1,49154
     755    1023    1243     749    1495    2984    2170
River Rch & RM= Dry Lacy Fork,Reach-1,48817
     942    1291    1580     960    1915    3820    2818
River Rch & RM= Dry Lacy Fork,Reach-1,47662
    1054    1451    1780    1083    2161    4311    3193
River Rch & RM= Dry Lacy Fork,Reach-1,44491
    1491    2072    2559    1564    3121    6226    4655
River Rch & RM= Dry Lacy Fork,Reach-1,38333
    1942    2729    3395    2089    4168    8316    6302
River Rch & RM= Dry Lacy Fork,Reach-1,36001
    2112    2977    3711    2288    4565    9109    6928
River Rch & RM= Dry Lacy Fork,Reach-1,35287
    2118    2984    3718    2291    4571    9121    6930
River Rch & RM= Dry Lacy Fork,Reach-1,33885
    2091    2933    3646    2240    4469    8917    6736
River Rch & RM= Dry Lacy Fork,Reach-1,30616
    2228    3132    3896    2396    4781    9540    7221
River Rch & RM= Dry Lacy Fork,Reach-1,28566
    2229    3131    3893    2392    4773    9524    7199
River Rch & RM= Dry Lacy Fork,Reach-1,26858
    2267    3184    3960    2434    4857    9690    7326
River Rch & RM= Dry Lacy Fork,Reach-1,26035
    2281    3199    3975    2440    4869    9715    7328
River Rch & RM= Dry Lacy Fork,Reach-1,21651
    2282    3199    3973    2438    4864    9706    7315
River Rch & RM= Dry Lacy Fork,Reach-1,20811
    2441    3431    4269    2624    5235   10445    7896
River Rch & RM= Dry Lacy Fork,Reach-1,19101
    2634    3705    4611    2834    5655   11284    8531
River Rch & RM= Dry Lacy Fork,Reach-1,13264
    2717    3823    4761    2928    5841   11655    8818
River Rch & RM= Dry Lacy Fork,Reach-1,11593
    2990    4207    5237    3217    6420   12809    9675
Boundary for River Rch & Prof#=Dry Lacy Fork,Reach-1,1
Up Type=0
Dn Type=3
Dn Slope=0.005
Boundary for River Rch & Prof#=Dry Lacy Fork,Reach-1,2
Up Type=0
Dn Type=3
Dn Slope=0.005
Boundary for River Rch & Prof#=Dry Lacy Fork,Reach-1,3
Up Type=0
Dn Type=3
Dn Slope=0.005
Boundary for River Rch & Prof#=Dry Lacy Fork,Reach-1,4
Up Type=0
Dn Type=3
Dn Slope=0.005
Boundary for River Rch & Prof#=Dry Lacy Fork,Reach-1,5
Up Type=0
Dn Type=3
Dn Slope=0.005
Boundary for River Rch & Prof#=Dry Lacy Fork,Reach-1,6
Up Type=0
Dn Type=3
Dn Slope=0.005
Boundary for River Rch & Prof#=Dry Lacy Fork,Reach-1,7
Up Type=0
Dn Type=3
Dn Slope=0.005

--- Dry Lacy Fork.g01 (geometry) ---

Geom Title=Existing Conditions

River Reach=Dry Lacy Fork,Reach-1
Reach XY= 30
      2767776.00      6901311.00      2766922.15      6898962.39
      2766081.82      6898363.31      2764768.60      6895505.23
      2762924.53      6894514.55      2761777.47      6894457.46
      2760933.74      6893567.46      2760599.52      6892083.88
      2758262.26      6891097.80      2756653.19      6888587.02
      2755173.46      6888155.70      2754786.17      6887521.33
      2753942.39      6887227.78      2753920.92      6886458.72
      2753126.49      6885750.55      2752983.52      6884961.05
      2753468.51      6884257.83      2753018.18      6883413.37
      2751469.94      6883402.86      2750020.32      6881212.97
      2748072.69      6880969.07      2747096.34      6881561.29
      2744733.98      6880857.78      2743970.04      6879663.14
      2740876.00      6879961.00      2739429.82      6878159.42
      2739273.77      6876516.90      2738570.39      6875116.59
      2734631.85      6874358.94      2734476.00      6873411.00

Type RM Length L Ch R = 1,58313,130,130,130
BEGIN DESCRIPTION:
Dry Lacy Fork 2864
END DESCRIPTION:
XS GIS Cut Line= 3
      2768087.67      6901283.55      2767775.90      6901279.19
      2767360.80      6901390.24
#Sta/Elev= 30
  4688.2  537.29  4719.9  536.40  4789.9  535.59  4799.9  535.31  4809.9  534.04
  4829.9  533.98  4839.9  533.31  4859.9  533.48  4869.9  533.26  4939.9  533.08
  4969.9  531.27  5010.2  530.82  5020.6  530.96  5026.1  530.52  5031.2  530.50
  5039.3  530.10  5039.6  529.60  5043.1  529.60  5043.3  530.10  5051.7  530.52
  5066.1  530.41  5082.7  530.82  5106.2  530.95  5124.1  531.60  5186.3  531.80
  5248.3  533.35  5261.2  533.35  5296.1  532.65  5320.8  532.44  5429.7  532.90
#Mann=3,-1,0
  4688.2    0.05       0  5039.3    0.04       0  5043.3    0.05       0
Bank Sta=5039.3,5043.3
Exp/Cntr=0.3,0.1

Type RM Length L Ch R = 1,58183,158,158,158
BEGIN DESCRIPTION:
Dry Lacy Fork 2862
END DESCRIPTION:
XS GIS Cut Line= 3
      2768066.05      6901151.39      2767719.59      6901165.35
      2767283.88      6901171.91
#Sta/Elev= 30
  4655.0  537.20  4725.1  535.94  4735.1  535.55  4745.1  534.97  4755.1  533.06
  4764.8  534.12  4775.1  533.81  4785.2  532.77  4795.2  533.11  4815.2  533.36
  4825.2  532.65  4905.3  531.73  4975.3  529.53  4993.3  529.41  4993.6  528.91
  4997.1  528.91  4997.3  529.41  5001.0  530.00  5006.0  530.00  5015.3  530.66
  5035.3  530.50  5055.3  530.61  5065.3  530.39  5125.3  531.08  5225.4  531.16
  5285.4  531.79  5345.4  532.08  5385.4  531.81  5415.4  532.13  5437.5  531.95
#Mann=3,-1,0
  4655.0    0.05       0  4993.3    0.04       0  4997.3    0.05       0
Bank Sta=4993.3,4997.3
Exp/Cntr=0.3,0.1

Type RM Length L Ch R = 1,58025,176,176,176
BEGIN DESCRIPTION:
Dry Lacy Fork 2861
END DESCRIPTION:
XS GIS Cut Line= 3
      2768051.93      6901007.31      2767673.27      6901022.20
      2767215.64      6901026.48
#Sta/Elev= 30
  4621.7  537.84  4627.6  537.36  4637.6  536.99  4667.7  536.51  4687.7  535.91
  4707.7  535.84  4727.7  535.10  4757.7  534.74  4827.8  532.23  4887.8  531.37
  4917.9  531.34  4927.9  530.40  4937.9  530.00  4957.9  529.79  4987.9  528.94
  4996.8  528.42  5005.9  528.41  5006.2  527.91  5009.7  527.91  5009.9  528.41
  5017.9  529.06  5077.9  529.44  5127.9  530.26  5197.9  530.57  5237.9  531.60
  5327.9  531.84  5367.9  531.32  5397.9  530.60  5417.9  531.09  5458.3  531.03
#Mann=3,-1,0
  4621.7    0.05       0  5005.9    0.04       0  5009.9    0.05       0
Bank Sta=5005.9,5009.9
Exp/Cntr=0.3,0.1

Type RM Length L Ch R = 1,57849,403,403,403
BEGIN DESCRIPTION:
Dry Lacy Fork 2863
END DESCRIPTION:
XS GIS Cut Line= 3
      2768052.96      6900848.01      2767622.98      6900861.63
      2767266.71      6900918.63
#Sta/Elev= 30
  4567.7  536.53  4614.7  535.35  4674.7  534.57  4724.7  533.20  4794.8  532.40
  4825.0  531.64  4864.8  531.55  4874.8  530.60  4884.8  530.16  4964.9  528.37
  4984.9  528.32  4993.9  527.59  4997.9  527.59  5003.0  526.93  5003.2  526.43
  5006.7  526.43  5007.0  526.93  5015.1  527.62  5065.7  528.29  5078.3  528.90
  5088.3  529.47  5136.6  529.81  5146.7  530.32  5197.4  530.47  5207.5  531.03
  5214.0  530.72  5219.1  530.95  5276.0  530.65  5281.1  531.01  5358.7  530.27
#Mann=5,-1,0
  4567.7    0.05       0  5003.0    0.04       0  5007.0    0.05       0
  5078.3    0.12       0  5088.3    0.05       0
Bank Sta=5003,5007
Exp/Cntr=0.3,0.1

Type RM Length L Ch R = 1,57446,172,172,172
BEGIN DESCRIPTION:
Dry Lacy Fork 2860
END DESCRIPTION:
XS GIS Cut Line= 3
      2767852.93      6900456.87      2767477.82      6900504.75
      2767169.35      6900650.45
#Sta/Elev= 30
  4624.2  533.20  4631.2  533.38  4641.3  535.02  4651.3  534.10  4661.4  531.86
  4682.0  531.07  4732.0  530.80  4742.1  529.89  4754.4  529.59  4782.2  529.32
  4812.6  528.95  4873.1  526.70  4903.4  526.66  4930.9  525.86  4936.0  525.21
  4953.8  525.37  4963.9  524.92  4973.9  523.69  4982.0  523.51  4982.3  523.01
  4985.8  523.01  4986.0  523.51  4994.1  524.65  5024.8  524.84  5073.0  526.17
  5081.8  526.72  5098.7  526.74  5104.2  527.14  5137.1  526.32  5343.5  527.47
#Mann=7,-1,0
  4624.2    0.05       0  4682.0    0.12       0  4754.4    0.05       0
  4782.2    0.12       0  4982.0    0.07       0  4986.0    0.12       0
  5073.0    0.05       0
Bank Sta=4982,4986
Exp/Cntr=0.3,0.1

Type RM Length L Ch R = 1,57274,288,288,288
BEGIN DESCRIPTION:
Dry Lacy Fork 2859
END DESCRIPTION:
XS GIS Cut Line= 3
      2767807.44      6900280.83      2767425.97      6900347.60
      2767069.22      6900492.19
#Sta/Elev= 30
  4611.4  531.29  4619.1  531.22  4673.8  530.46  4704.4  529.27  4724.5  529.19
  4753.7  528.37  4765.1  528.52  4785.4  527.61  4795.6  526.66  4818.2  526.35
  4836.2  525.58  4877.6  524.60  4917.4  524.26  4926.9  523.87  4947.9  524.03
  4968.2  523.33  4986.4  523.25  4991.5  523.04  4994.1  521.83  4994.4  521.33
  4997.9  521.33  4998.1  521.83  5001.3  521.83  5031.0  524.17  5041.8  524.34
  5076.9  526.01  5085.6  525.92  5202.8  524.99  5310.0  525.97  5383.6  525.89
#Mann=5,-1,0
  4611.4    0.05       0  4619.1    0.12       0  4994.1    0.07       0
  4998.1    0.12       0  5085.6    0.05       0
Bank Sta=4994.1,4998.1
Exp/Cntr=0.3,0.1

Type RM Length L Ch R = 1,56986,212,212,212
BEGIN DESCRIPTION:
Dry Lacy Fork 2858
END DESCRIPTION:
XS GIS Cut Line= 3
      2767699.49      6900020.12      2767325.27      6900090.54
      2766948.08      6900356.30
#Sta/Elev= 30
  4621.4  528.14  4686.2  526.95  4808.1  524.70  4838.6  525.38  4859.0  524.88
  4879.3  524.03  4899.7  523.72  4924.4  522.84  4930.2  522.94  4976.8  520.09
  4981.9  520.86  4991.3  520.87  4999.3  519.97  5009.5  520.22  5013.7  518.64
  5013.9  518.14  5017.4  518.14  5017.7  518.64  5024.3  519.38  5030.5  520.45
  5038.0  522.37  5045.3  523.76  5051.4  524.40  5060.1  524.06  5074.7  522.56
  5131.5  522.63  5137.6  522.45  5274.3  524.24  5390.1  524.19  5463.6  525.14
#Mann=4,-1,0
  4621.4    0.12       0  4686.2    0.05       0  5013.7    0.05       0
  5017.7    0.05       0
Bank Sta=5013.7,5017.7
Exp/Cntr=0.3,0.1

Type RM Length L Ch R = 1,56774,222,222,222
BEGIN DESCRIPTION:
Dry Lacy Fork 2857
END DESCRIPTION:
XS GIS Cut Line= 3
      2767670.28      6899776.95      2767227.04      6899911.47
      2766908.51      6900286.16
#Sta/Elev= 30
  4535.6  526.99  4550.5  526.34  4561.0  526.55  4604.6  525.92  4703.3  523.61
  4822.2  522.48  4911.1  520.73  4916.3  520.99  4944.0  520.36  4949.2  520.71
  5001.8  518.70  5006.4  517.52  5011.0  517.00  5011.3  516.50  5014.8  516.50
  5015.0  517.00  5020.7  518.89  5027.3  519.52  5049.3  520.24  5070.1  520.11
  5098.7  520.96  5119.5  520.74  5176.7  522.27  5183.2  521.98  5191.0  522.37
  5211.8  522.21  5297.5  523.39  5339.4  522.95  5382.0  523.27  5490.6  525.03
#Mann=3,-1,0
  4535.6    0.05       0  5011.0    0.04       0  5015.0    0.05       0
Bank Sta=5011,5015
Exp/Cntr=0.3,0.1

Type RM Length L Ch R = 1,56552,441,441,441
BEGIN DESCRIPTION:
Dry Lacy Fork 2856
END DESCRIPTION:
XS GIS Cut Line= 3
      2767655.27      6899731.54      2767171.95      6899707.48
      2766781.49      6899796.10
#Sta/Elev= 30
  4519.1  524.92  4558.4  525.62  4588.5  524.56  4638.5  523.49  4788.7  521.02
  4808.7  521.06  4868.8  519.66  4888.8  519.70  4918.9  518.87  4938.9  518.75
  4968.9  517.26  4988.9  517.96  4998.5  516.47  5003.0  516.47  5009.1  515.60
  5017.4  515.51  5017.6  515.01  5021.1  515.01  5021.4  515.51  5029.6  516.93
  5043.2  517.69  5050.1  517.43  5086.3  518.30  5101.4  518.16  5129.4  519.18
  5134.6  518.93  5152.7  519.32  5255.2  518.90  5360.3  520.31  5403.4  520.29
#Mann=3,-1,0
  4519.1    0.05       0  5017.4    0.04       0  5021.4    0.05       0
Bank Sta=5017.4,5021.4
Exp/Cntr=0.3,0.1

Type RM Length L Ch R = 1,56111,307,307,307
BEGIN DESCRIPTION:
Dry Lacy Fork 2855
END DESCRIPTION:
XS GIS Cut Line= 3
      2767624.46      6899377.49      2767075.00      6899298.11
      2766704.57      6899391.16
#Sta/Elev= 30
  4446.0  522.43  4460.7  522.11  4495.0  521.78  4528.3  521.00  4565.7  521.02
  4697.0  519.65  4828.4  517.83  4875.0  516.82  4899.1  516.84  4919.3  515.89
  4945.3  513.73  4969.8  513.56  4979.9  513.96  5003.2  513.74  5010.4  513.46
  5018.8  512.36  5019.0  511.86  5022.5  511.86  5022.8  512.36  5051.7  513.61
  5062.0  513.47  5070.9  513.83  5076.0  514.22  5082.6  515.39  5117.2  515.26
  5144.5  515.95  5194.3  516.02  5247.6  517.17  5309.5  516.78  5383.1  517.91
#Mann=4,-1,0
  4446.0    0.12       0  4460.7    0.05       0  5018.8    0.05       0
  5022.8    0.05       0
Bank Sta=5018.8,5022.8
Exp/Cntr=0.3,0.1

Type RM Length L Ch R = 1,55804,353,353,353
BEGIN DESCRIPTION:
Dry Lacy Fork 2854
END DESCRIPTION:
XS GIS Cut Line= 3
      2767288.22      6898799.42      2766942.22      6899033.33
      2766688.03      6899350.88
#Sta/Elev= 30
  4587.1  520.86  4591.5  520.86  4597.3  519.82  4616.4  519.28  4648.3  519.42
  4720.2  518.97  4747.2  519.15  4783.2  518.58  4792.1  517.94  4813.1  517.06
  4834.1  516.72  4906.0  514.35  4921.0  513.55  4935.9  512.18  4977.9  511.86
  4990.9  511.12  4991.2  510.62  4994.7  510.62  4994.9  511.12  5007.4  511.77
  5028.2  511.80  5050.6  513.39  5057.1  513.10  5065.1  513.32  5085.9  512.93
  5100.3  513.01  5149.9  514.01  5263.5  514.75  5356.4  516.79  5411.5  517.29
#Mann=4,-1,0
  4587.1    0.12       0  4616.4    0.05       0  4990.9    0.04       0
  4994.9    0.05       0
Bank Sta=4990.9,4994.9
Exp/Cntr=0.3,0.1

Type RM Length L Ch R = 1,55451,638,638,638
BEGIN DESCRIPTION:
Dry Lacy Fork 2782
END DESCRIPTION:
XS GIS Cut Line= 3
      2766969.67      6898542.84      2766644.50      6898882.93
      2766591.86      6899236.81
#Sta/Elev= 30
  4603.8  516.53  4683.0  515.05  4795.9  512.05  4838.4  511.63  4845.6  511.96
  4859.8  511.97  4880.8  511.31  4937.5  511.45  4979.9  510.00  4992.1  509.05
  4992.3  508.55  4995.8  508.55  4996.1  509.05  5008.2  509.21  5015.5  509.97
  5022.4  510.11  5050.7  509.92  5057.8  510.01  5064.8  510.53  5074.3  510.52
  5097.9  512.52  5122.9  513.15  5167.2  513.45  5203.8  513.16  5244.2  513.33
  5254.4  513.97  5264.5  514.10  5274.6  513.72  5284.7  513.78  5432.1  515.61
#Mann=3,-1,0
  4603.8    0.05       0  4992.1    0.04       0  4996.1    0.05       0
Bank Sta=4992.1,4996.1
Exp/Cntr=0.3,0.1

Type RM Length L Ch R = 1,54813,284,284,284
BEGIN DESCRIPTION:
Dry Lacy Fork 2830
END DESCRIPTION:
XS GIS Cut Line= 3
      2766505.82      6898268.68      2766277.92      6898499.78
      2765809.51      6898818.44
#Sta/Elev= 30
  4669.1  511.37  4720.1  511.25  4769.7  509.87  4783.8  510.07  4847.4  509.33
  4896.9  507.94  4939.3  507.98  4953.4  507.69  4960.5  506.97  4967.6  507.07
  4974.7  506.33  5003.4  506.62  5016.3  506.28  5016.6  505.78  5020.1  505.78
  5020.3  506.28  5024.4  508.07  5039.3  508.62  5045.4  509.36  5090.2  509.25
  5111.1  510.30  5162.0  511.66  5176.9  512.57  5183.0  512.23  5225.8  512.94
  5239.9  513.61  5334.6  514.38  5362.6  515.10  5377.5  516.06  5560.2  518.50
#Mann=3,-1,0
  4669.1    0.05       0  5016.3    0.05       0  5020.3    0.05       0
Bank Sta=5016.3,5020.3
Exp/Cntr=0.3,0.1

Type RM Length L Ch R = 1,54529,136,136,136
BEGIN DESCRIPTION:
Dry Lacy Fork 2780
END DESCRIPTION:
XS GIS Cut Line= 3
      2766497.02      6898253.33      2766074.69      6898323.36
      2765595.30      6898405.06
#Sta/Elev= 30
  4570.3  511.39  4611.9  511.19  4662.6  510.26  4682.8  509.38  4708.5  509.06
  4830.5  508.18  4865.3  507.56  4946.4  507.23  4976.8  506.56  4998.4  506.91
  5025.5  505.85  5025.8  505.35  5029.3  505.35  5029.5  505.85  5037.6  506.67
  5057.9  506.86  5078.5  508.13  5118.8  508.09  5139.1  509.32  5179.7  510.57
  5188.7  511.27  5230.4  512.30  5248.9  513.19  5254.0  512.94  5321.7  514.53
  5331.8  514.14  5369.3  514.16  5463.7  515.38  5473.8  515.95  5484.7  515.92
#Mann=3,-1,0
  4570.3    0.05       0  5025.5    0.05       0  5029.5    0.05       0
Bank Sta=5025.5,5029.5
Exp/Cntr=0.3,0.1

Type RM Length L Ch R = 1,54393,656,656,656
BEGIN DESCRIPTION:
Dry Lacy Fork 2779
END DESCRIPTION:
XS GIS Cut Line= 4
      2766463.98      6897995.27      2766104.65      6898200.95
      2766021.14      6898202.54      2765514.14      6898244.60
#Sta/Elev= 30
  4507.8  512.46  4510.3  513.36  4526.1  512.66  4540.0  512.75  4547.7  512.01
  4649.8  510.91  4655.6  511.88  4665.7  511.01  4678.3  511.37  4708.8  509.67
  4730.4  509.29  4736.2  509.63  4746.3  508.92  4773.6  508.85  4826.8  507.44
  4980.5  507.37  5000.4  505.40  5008.5  505.26  5008.8  504.76  5012.3  504.76
  5012.5  505.26  5030.6  507.59  5040.6  506.92  5080.8  508.16  5292.8  510.65
  5381.8  513.58  5401.9  515.00  5413.5  514.62  5421.9  515.22  5514.1  516.44
#Mann=3,-1,0
  4507.8    0.05       0  5008.5    0.05       0  5012.5    0.05       0
Bank Sta=5008.5,5012.5
Exp/Cntr=0.3,0.1

Type RM Length L Ch R = 1,53737,398,398,398
BEGIN DESCRIPTION:
Dry Lacy Fork 2728
END DESCRIPTION:
XS GIS Cut Line= 3
      2766391.58      6897519.20      2765975.77      6897609.40
      2765329.61      6897939.10
#Sta/Elev= 30
  4575.3  516.42  4621.9  515.75  4642.4  514.77  4765.2  505.98  4842.6  504.10
  4898.2  504.35  4918.7  503.65  4985.0  503.45  4998.1  501.76  5008.7  501.45
  5009.0  500.95  5012.7  501.45  5032.9  503.70  5067.9  504.06  5127.5  506.32
  5188.5  505.84  5247.5  507.98  5327.5  508.33  5344.1  508.61  5349.7  509.50
  5359.8  508.90  5449.6  509.63  5477.5  510.28  5483.3  512.48  5494.1  512.75
  5499.7  510.73  5505.7  510.64  5618.0  512.69  5662.9  512.79  5726.2  514.32
#Mann=3,-1,0
  4575.3    0.05       0  5008.7    0.04       0  5012.7    0.05       0
Bank Sta=5008.7,5012.7
Exp/Cntr=0.3,0.1

Type RM Length L Ch R = 1,53339,672,672,672
BEGIN DESCRIPTION:
Dry Lacy Fork 2729
END DESCRIPTION:
XS GIS Cut Line= 3
      2766306.43      6897402.80      2765807.82      6897283.14
      2765107.21      6897622.65
#Sta/Elev= 30
  4404.8  514.25  4456.7  511.52  4516.4  507.10  4558.4  505.14  4610.9  504.38
  4631.5  503.35  4694.7  503.13  4754.9  502.03  4820.7  501.66  4847.4  501.94
  4952.9  501.11  4964.0  501.43  4990.4  499.77  4990.6  499.27  4994.1  499.27
  4994.4  499.77  4997.9  500.54  5043.1  501.57  5060.1  501.31  5088.2  502.26
  5105.3  501.68  5127.8  501.75  5133.4  502.50  5164.1  503.38  5178.5  504.38
  5246.3  506.47  5308.5  505.79  5359.2  505.94  5553.0  508.85  5696.1  509.83
#Mann=3,-1,0
  4404.8    0.05       0  4990.4    0.04       0  4994.4    0.05       0
Bank Sta=4990.4,4994.4
Exp/Cntr=0.3,0.1

Type RM Length L Ch R = 1,52667,639,639,639
BEGIN DESCRIPTION:
Dry Lacy Fork 2727
END DESCRIPTION:
XS GIS Cut Line= 3
      2766091.90      6896704.80      2765331.61      6896848.85
      2764856.84      6897190.44
#Sta/Elev= 30
  4271.2  510.39  4332.3  509.66  4379.0  507.28  4419.7  503.54  4460.4  501.57
  4592.7  499.31  4651.2  499.43  4656.3  499.85  4806.5  499.42  4813.2  499.00
  4857.3  499.47  4870.6  498.59  4928.6  497.77  4969.3  497.90  4973.2  495.55
  4973.4  495.05  4976.9  495.05  4977.2  495.55  4980.3  496.04  4989.7  495.78
  4999.8  498.05  5020.2  498.86  5051.5  498.82  5072.4  499.95  5128.9  500.11
  5223.4  501.40  5250.4  502.56  5279.8  502.42  5401.4  504.16  5629.9  505.64
#Mann=3,-1,0
  4271.2    0.05       0  4973.2    0.05       0  4977.2    0.05       0
Bank Sta=4973.2,4977.2
Exp/Cntr=0.3,0.1

Type RM Length L Ch R = 1,52028,448,448,448
BEGIN DESCRIPTION:
Dry Lacy Fork 2724
END DESCRIPTION:
XS GIS Cut Line= 3
      2765841.00      6896054.39      2765241.46      6896340.93
      2764920.89      6896734.76
#Sta/Elev= 30
  4346.1  516.27  4444.2  511.35  4557.6  502.88  4563.2  504.02  4625.6  502.57
  4653.9  504.36  4728.5  497.76  4927.1  496.31  4948.7  490.62  4954.2  494.00
  4971.4  491.87  4976.9  494.51  4981.3  490.41  4981.6  489.91  4985.5  490.41
  4999.6  490.70  5010.6  492.61  5014.2  494.92  5022.1  491.95  5028.6  496.12
  5036.5  495.31  5043.0  492.62  5049.4  495.40  5057.3  491.67  5063.8  496.87
  5071.7  496.30  5078.1  499.05  5216.8  500.51  5313.0  499.87  5518.4  502.42
#Mann=5,-1,0
  4346.1    0.05       0  4927.1    0.12       0  4981.3    0.07       0
  4985.5    0.12       0  5216.8    0.05       0
Bank Sta=4981.3,4985.5
Exp/Cntr=0.3,0.1

Type RM Length L Ch R = 1,51580,464,464,464
BEGIN DESCRIPTION:
Dry Lacy Fork 2726
END DESCRIPTION:
XS GIS Cut Line= 3
      2765603.44      6895459.67      2765050.55      6895993.33
      2764761.08      6896486.07
#Sta/Elev= 30
  4237.6  520.95  4342.9  515.88  4420.6  511.03  4470.2  506.54  4547.9  502.62
  4682.2  497.85  4807.5  495.75  4901.4  495.31  4958.0  492.83  4965.2  494.38
  4979.3  494.43  4986.3  493.24  5000.4  493.94  5005.7  492.84  5022.8  494.42
  5038.1  490.95  5042.1  488.32  5042.5  487.82  5046.4  488.32  5059.9  494.43
  5065.7  496.13  5087.2  496.19  5102.9  495.09  5124.3  496.16  5154.1  495.71
  5219.1  497.11  5518.9  501.72  5556.1  504.47  5571.6  504.56  5577.5  503.05
#Mann=5,-1,0
  4237.6    0.05       0  4807.5    0.12       0  5042.1    0.07       0
  5046.4    0.12       0  5219.1    0.05       0
Bank Sta=5042.1,5046.4
Exp/Cntr=0.3,0.1

Type RM Length L Ch R = 1,51116,416,416,416
BEGIN DESCRIPTION:
Dry Lacy Fork 2725
END DESCRIPTION:
XS GIS Cut Line= 3
      2765272.08      6895216.01      2764762.57      6895657.20
      2764525.85      6896007.06
#Sta/Elev= 30
  4333.3  519.11  4376.8  518.58  4419.5  515.98  4426.1  514.95  4497.4  511.36
  4561.0  507.24  4610.4  502.61  4681.7  498.09  4773.8  494.94  4882.6  493.58
  4901.0  493.38  4908.7  491.84  4922.9  491.23  4929.5  493.00  4978.9  492.00
  4986.5  490.20  4993.2  486.89  4998.6  486.71  4999.0  486.21  5003.0  486.71
  5022.9  493.67  5071.2  495.25  5085.9  495.94  5144.7  495.39  5208.7  495.87
  5259.6  497.75  5325.5  498.99  5331.6  499.80  5388.5  499.58  5429.7  500.29
#Mann=5,-1,0
  4333.3    0.05       0  4882.6    0.12       0  4998.6    0.07       0
  5003.0    0.12       0  5071.2    0.05       0
Bank Sta=4998.6,5003
Exp/Cntr=0.3,0.1

Type RM Length L Ch R = 1,50700,770,770,770
BEGIN DESCRIPTION:
Dry Lacy Fork 2666
END DESCRIPTION:
XS GIS Cut Line= 3
      2765106.91      6894949.10      2764601.48      6895357.92
      2764230.83      6895824.42
#Sta/Elev= 30
  4364.5  514.22  4466.5  512.54  4472.9  513.38  4480.9  511.61  4487.3  512.43
  4536.9  505.30  4615.2  502.24  4629.6  500.56  4672.8  498.26  4800.7  493.96
  4893.0  492.31  4914.2  491.01  4921.7  491.55  4963.8  491.86  4978.2  487.67
  4990.3  486.96  4990.7  486.46  4994.7  486.96  5006.9  491.07  5028.2  492.67
  5063.4  491.95  5076.9  490.20  5092.2  489.64  5098.6  491.09  5106.7  491.01
  5113.0  492.62  5191.6  495.92  5276.4  495.17  5497.5  499.34  5610.4  500.13
#Mann=5,-1,0
  4364.5    0.05       0  4921.7    0.12       0  4990.3    0.07       0
  4994.7    0.12       0  5076.9    0.05       0
Bank Sta=4990.3,4994.7
Exp/Cntr=0.3,0.1

Type RM Length L Ch R = 1,49930,776,776,776
BEGIN DESCRIPTION:
Dry Lacy Fork 2665
END DESCRIPTION:
XS GIS Cut Line= 3
      2764328.58      6894660.25      2763940.58      6895096.18
      2763698.73      6895767.56
#Sta/Elev= 30
  4460.5  499.47  4547.8  498.53  4582.9  498.83  4590.5  499.48  4660.9  496.55
  4698.3  494.06  4746.0  491.92  4796.1  487.66  4843.2  487.03  4843.7  486.53
  4847.7  487.03  4873.9  488.99  4923.2  488.55  4937.5  489.20  4965.9  488.06
  4994.3  489.01  5043.7  488.35  5059.8  488.95  5081.1  488.10  5091.7  488.73
  5186.2  488.94  5272.4  490.25  5339.7  492.33  5365.1  493.81  5370.4  493.41
  5463.7  496.05  5600.0  496.58  5612.6  495.77  5623.2  497.26  5757.7  497.62
#Mann=5,-1,0
  4460.5    0.05       0  4660.9     0.1       0  4698.3    0.05       0
  4843.2    0.04       0  4847.7    0.05       0
Bank Sta=4843.2,4847.7
Exp/Cntr=0.3,0.1

Type RM Length L Ch R = 1,49154,337,337,337
BEGIN DESCRIPTION:
Dry Lacy Fork 2664
END DESCRIPTION:
XS GIS Cut Line= 3
      2763853.35      6893842.34      2763280.57      6894798.11
      2763337.40      6895581.29
#Sta/Elev= 30
  3945.6  502.19  3955.8  502.87  3971.4  501.92  4014.2  501.18  4305.8  499.70
  4342.7  499.11  4358.3  498.05  4387.1  498.22  4395.2  496.79  4527.0  491.42
  4533.3  489.60  4561.9  486.24  4766.6  486.45  4898.8  485.49  4935.0  486.08
  4984.3  485.51  4997.6  484.09  4998.1  483.59  5002.1  484.09  5005.7  485.63
  5021.3  486.43  5143.0  486.43  5313.4  488.06  5413.7  490.97  5479.6  494.03
  5574.1  495.64  5753.1  496.73  5758.1  496.19  5774.6  496.85  5845.1  495.93
#Mann=3,-1,0
  3945.6    0.05       0  4997.6    0.04       0  5002.1    0.05       0
Bank Sta=4997.6,5002.1
Exp/Cntr=0.3,0.1

Type RM Length L Ch R = 1,48817,486,486,486
BEGIN DESCRIPTION:
Dry Lacy Fork 27
END DESCRIPTION:
XS GIS Cut Line= 3
      2763004.07      6893701.58      2763026.00      6894611.00
      2762653.95      6895866.86
#Sta/Elev= 30
  4094.8  504.18  4154.2  502.60  4194.3  503.84  4234.3  501.26  4334.3  497.54
  4354.3  498.09  4364.3  496.75  4514.3  491.36  4537.9  489.58  4646.1  487.39
  4944.5  484.63  4971.8  483.06  4972.6  482.56  4977.1  483.06  4994.5  484.88
  5119.2  486.03  5380.0  493.89  5512.6  489.09  5578.1  485.38  5745.0  486.34
  5776.3  488.02  5891.0  490.31  5899.2  490.67  5911.9  493.46  5976.1  492.84
  5984.9  494.02  6081.1  496.58  6109.1  496.24  6147.6  497.95  6314.3  501.21
#Mann=5,-1,0
  4094.8    0.05       0  4537.9    0.12       0  4646.1    0.05       0
  4971.8    0.04       0  4977.1    0.05       0
Bank Sta=4971.8,4977.1
Exp/Cntr=0.3,0.1

Type RM Length L Ch R = 1,48331,484,484,484
BEGIN DESCRIPTION:
Dry Lacy Fork 26
END DESCRIPTION:
XS GIS Cut Line= 3
      2762576.91      6893759.87      2762576.00      6894511.00
      2762576.00      6895710.97
#Sta/Elev= 30
  4248.9  513.48  4320.0  512.20  4366.4  509.51  4380.0  508.99  4470.0  500.22
  4490.0  500.37  4500.0  499.32  4520.0  495.69  4600.0  491.38  4660.0  488.99
  4690.0  489.02  4780.0  486.23  4832.3  486.69  4850.0  486.33  4880.0  483.17
  4929.6  484.27  5007.3  483.00  5008.1  482.50  5012.7  483.00  5060.0  483.67
  5230.0  483.21  5456.3  483.89  5530.0  485.28  5610.0  485.70  5710.0  488.69
  5780.0  489.17  5830.0  491.47  6000.0  495.54  6120.0  497.45  6200.0  500.01
#Mann=7,-1,0
  4248.9    0.05       0  4366.4    0.12       0  4832.3    0.05       0
  4929.6    0.12       0  5007.3    0.07       0  5012.7    0.12       0
  5456.3    0.05       0
Bank Sta=5007.3,5012.7
Exp/Cntr=0.3,0.1

Type RM Length L Ch R = 1,47847,185,185,185
BEGIN DESCRIPTION:
Dry Lacy Fork 25
END DESCRIPTION:
XS GIS Cut Line= 3
      2762481.31      6893710.72      2762126.00      6894511.00
      2762525.99      6895710.97
#Sta/Elev= 30
  4119.6  510.52  4192.7  508.98  4221.4  507.09  4239.2  507.53  4273.4  506.05
  4291.2  506.28  4296.7  505.10  4360.6  502.99  4371.9  501.38  4488.2  495.14
  4685.3  486.36  4693.9  486.86  4783.8  483.29  4827.0  482.85  4828.0  482.35
  4833.7  482.85  5307.9  483.41  5414.0  485.71  5519.6  488.04  5585.5  490.47
  5606.6  490.07  5669.8  492.05  5680.4  491.58  5782.2  493.17  5901.7  494.57
  5943.9  493.12  5986.1  493.26  6028.2  495.19  6175.8  497.67  6260.1  500.09
#Mann=8,-1,0
  4119.6    0.12       0  4693.9    0.05       0  4827.0    0.03       0
  4833.7    0.05       0  5307.9    0.12       0  5414.0     0.1       0
  5519.6    0.12       0  5782.2    0.05       0
Bank Sta=4827,4833.7
Exp/Cntr=0.3,0.1

Type RM Length L Ch R = 1,47662,584,584,584
BEGIN DESCRIPTION:
Dry Lacy Fork 2637
END DESCRIPTION:
XS GIS Cut Line= 3
      2762422.16      6893610.56      2761946.92      6894493.92
      2761017.45      6895810.13
#Sta/Elev= 30
  4005.6  512.62  4152.8  506.29  4239.6  504.38  4349.1  500.43  4387.2  497.60
  4425.4  496.74  4512.0  492.50  4742.7  483.81  4832.3  482.85  4833.4  482.35
  4839.7  482.85  5273.7  482.89  5315.5  483.53  5353.8  485.28  5466.9  490.57
  5508.8  489.77  5553.1  490.22  5624.5  487.98  5630.6  486.98  5666.3  489.10
  5796.9  491.72  5811.7  492.34  5817.8  494.25  5832.6  494.15  5838.7  492.95
  5853.5  492.18  5947.7  492.01  6053.9  493.48  6278.3  495.59  6620.0  500.82
#Mann=7,-1,0
  4005.6    0.05       0  4152.8    0.12       0  4512.0    0.05       0
  4832.3    0.03       0  4839.7    0.05       0  5353.8    0.12       0
  6053.9    0.05       0
Bank Sta=4832.3,4839.7
Exp/Cntr=0.3,0.1

Type RM Length L Ch R = 1,47078,554,554,554
BEGIN DESCRIPTION:
Dry Lacy Fork 2636
END DESCRIPTION:
XS GIS Cut Line= 3
      2762489.75      6893368.01      2761698.23      6893883.75
      2760774.16      6895326.10
#Sta/Elev= 30
  3729.6  509.20  3820.6  509.94  3871.9  509.75  3893.0  510.33  3923.2  509.91
  3986.5  510.39  4104.1  509.08  4211.5  504.59  4327.6  497.60  4421.2  492.73
  4442.3  491.11  4457.4  490.91  4478.5  489.50  4499.6  488.83  4581.2  484.08
  4623.4  483.09  5177.9  482.78  5179.1  482.28  5184.4  482.28  5185.5  482.78
  5448.4  482.91  5536.3  486.40  5574.0  487.10  5614.9  487.79  5636.0  488.90
  5694.9  489.46  6057.1  494.76  6202.5  497.47  6317.5  500.90  6387.3  501.46
#Mann=5,-1,0
  3729.6    0.05       0  5177.9    0.03       0  5185.5    0.05       0
  5574.0    0.12       0  5694.9    0.05       0
Bank Sta=5177.9,5185.5
Exp/Cntr=0.3,0.1

Type RM Length L Ch R = 1,46524,122,122,122
BEGIN DESCRIPTION:
Dry Lacy Fork 2550
END DESCRIPTION:
XS GIS Cut Line= 3
      2762486.55      6893316.01      2761390.49      6893562.01
      2760622.14      6895062.72
#Sta/Elev= 30
  3754.0  507.60  3940.4  507.23  4032.2  506.22  4118.8  503.97  4210.6  503.76
  4259.1  502.69  4350.9  499.41  4437.5  494.54  4502.7  492.37  4554.0  488.27
  4605.2  486.31  4646.2  482.91  5254.3  482.79  5255.4  482.29  5262.1  482.79
  5505.3  482.88  5628.9  486.30  5756.0  487.28  5772.6  489.18  5786.2  487.31
  5794.8  487.20  5965.9  488.86  6255.5  494.33  6322.1  496.67  6327.7  498.80
  6394.4  498.12  6455.4  499.33  6461.0  500.36  6471.5  500.64  6563.3  499.77
#Mann=3,-1,0
  3754.0    0.05       0  5254.3    0.03       0  5262.1    0.05       0
Bank Sta=5254.3,5262.1
Exp/Cntr=0.3,0.1

Type RM Length L Ch R = 1,46402,161,161,161
BEGIN DESCRIPTION:
Dry Lacy Fork 2549
END DESCRIPTION:
XS GIS Cut Line= 3
      2761749.58      6892674.62      2761463.71      6893117.86
      2760601.02      6895003.78
#Sta/Elev= 30
  3875.1  505.60  4040.9  503.98  4049.3  505.73  4077.2  500.84  4092.4  493.66
  4124.8  492.60  4126.0  492.10  4132.6  492.60  4316.2  494.97  4382.5  499.33
  4427.8  499.19  4433.3  496.89  4456.3  499.24  4576.9  499.71  5708.1  499.64
  5731.1  497.25  5736.6  499.49  5754.2  497.90  5857.5  499.46  5874.7  497.37
  5880.2  499.55  5920.8  497.84  5978.5  499.25  5995.3  496.83  6000.8  499.16
  6018.3  496.53  6023.8  499.19  6161.9  499.01  6213.5  495.34  6476.4  500.98
#Mann=3,-1,0
  3875.1    0.05       0  4124.8    0.04       0  4132.6    0.05       0
Bank Sta=4124.8,4132.6
Exp/Cntr=0.3,0.1

Type RM Length L Ch R = 1,46241,337,337,337
BEGIN DESCRIPTION:
Dry Lacy Fork 2551
END DESCRIPTION:
XS GIS Cut Line= 3
      2761325.28      6892781.11      2761253.34      6893173.32
      2760641.41      6894656.16
#Sta/Elev= 30
  4092.1  487.79  4183.5  486.61  4196.7  488.71  4203.8  489.08  4222.9  484.74
  4234.3  483.71  4407.2  480.44  4437.7  480.31  4445.6  481.73  4450.6  480.79
  4458.0  482.43  4495.4  478.50  4542.4  476.45  4785.6  476.65  4945.4  474.27
  4953.5  472.30  5042.6  472.19  5043.7  471.69  5050.4  472.19  5051.9  474.58
  5061.7  476.80  5083.3  476.36  5206.3  479.39  5213.2  481.08  5224.0  480.12
  5437.8  485.89  5626.9  486.96  5650.9  486.30  5851.4  488.50  6095.0  493.73
#Mann=4,-1,0
  4092.1    0.12       0  4196.7    0.05       0  5042.6    0.04       0
  5050.4    0.05       0
Bank Sta=5042.6,5050.4
Exp/Cntr=0.3,0.1

Type RM Length L Ch R = 1,45904,684,684,684
BEGIN DESCRIPTION:
Dry Lacy Fork 2552
END DESCRIPTION:
XS GIS Cut Line= 3
      2761436.23      6892593.30      2760862.40      6893414.85
      2760416.24      6894437.33
#Sta/Elev= 30
  4010.4  495.87  4077.8  494.12  4239.4  486.96  4388.3  483.07  4397.8  484.56
  4410.1  483.81  4433.5  479.88  4654.2  475.99  4755.4  475.82  4799.9  473.50
  4820.8  475.34  4871.1  475.53  4928.1  475.72  4963.8  474.99  4978.7  472.45
  5004.9  473.13  5012.5  473.42  5016.4  471.90  5017.6  471.40  5024.3  471.90
  5052.0  475.86  5195.1  476.31  5218.6  475.10  5242.0  476.12  5259.3  474.89
  5411.3  477.96  5433.8  476.48  5690.7  486.39  5881.2  486.95  6128.1  490.26
#Mann=7,-1,0
  4010.4    0.05       0  4077.8    0.12       0  4388.3    0.05       0
  4871.1    0.12       0  5004.9    0.05       0  5016.4    0.07       0
  5024.3    0.05       0
Bank Sta=5016.4,5024.3
Exp/Cntr=0.3,0.1

Type RM Length L Ch R = 1,45220,239,239,239
BEGIN DESCRIPTION:
Dry Lacy Fork 2554
END DESCRIPTION:
XS GIS Cut Line= 3
      2761497.42      6892513.27      2760873.25      6892821.97
      2760131.56      6893466.13
#Sta/Elev= 30
  4313.6  496.71  4442.4  493.25  4516.0  491.61  4672.1  483.87  4684.8  482.31
  4746.5  479.83  4895.3  474.98  4939.9  470.45  4948.4  471.55  4962.2  469.83
  4970.9  470.51  4980.6  469.64  4981.8  469.14  4988.5  469.64  4993.3  470.57
  4998.9  473.37  5005.6  473.42  5057.2  471.72  5078.1  472.55  5085.7  473.78
  5092.4  472.54  5113.2  472.50  5170.2  474.51  5241.5  473.86  5276.6  475.01
  5347.8  473.15  5630.8  473.96  5794.1  478.74  5836.8  480.97  5992.3  482.34
#Mann=5,-1,0
  4313.6    0.05       0  4442.4    0.12       0  4672.1    0.05       0
  4980.6    0.04       0  4988.5    0.05       0
Bank Sta=4980.6,4988.5
Exp/Cntr=0.3,0.1

Type RM Length L Ch R = 1,44981,490,490,490
BEGIN DESCRIPTION:
Dry Lacy Fork 2553
END DESCRIPTION:
XS GIS Cut Line= 3
      2761524.48      6892486.21      2760838.53      6892587.17
      2760171.26      6893216.25
#Sta/Elev= 30
  4289.7  497.15  4439.7  492.61  4510.5  491.61  4559.5  488.28  4666.9  483.17
  4682.4  482.83  4712.7  480.50  4833.3  476.49  4988.2  474.61  5008.8  472.81
  5019.0  469.00  5020.2  468.50  5026.9  469.00  5037.1  471.56  5065.5  474.18
  5107.9  472.22  5129.0  472.27  5150.4  474.01  5192.7  473.27  5277.4  473.60
  5433.2  471.78  5482.6  473.76  5504.0  472.56  5546.5  472.47  5567.5  472.86
  5589.0  474.99  5680.8  477.80  5730.2  478.24  5829.3  481.08  5900.1  481.64
#Mann=5,-1,0
  4289.7    0.05       0  4439.7    0.12       0  4666.9    0.05       0
  5019.0    0.04       0  5026.9    0.05       0
Bank Sta=5019,5026.9
Exp/Cntr=0.3,0.1

Type RM Length L Ch R = 1,44491,1891,1891,1891
BEGIN DESCRIPTION:
Dry Lacy Fork 3462
END DESCRIPTION:
XS GIS Cut Line= 3
      2761485.99      6892381.35      2760712.65      6892216.94
      2758842.01      6892777.33
#Sta/Elev= 30
  4221.6  494.44  4291.7  492.01  4296.8  490.78  4348.6  489.99  4435.4  487.06
  4487.6  484.12  4589.6  479.32  4727.9  475.07  4871.6  473.19  4988.4  473.35
  5012.2  471.53  5015.2  469.01  5016.4  468.51  5023.2  469.01  5039.3  471.18
  5071.4  473.18  5520.2  471.52  5638.2  472.33  5749.9  475.57  5802.1  475.86
  6010.9  475.47  6050.9  474.48  6089.2  471.76  6136.1  471.41  6364.3  472.28
  6501.5  475.77  6512.3  477.31  6749.1  485.29  6924.9  490.08  6965.0  489.92
#Mann=5,-1,0
  4221.6    0.05       0  4348.6    0.12       0  4487.6    0.05       0
  5015.2    0.04       0  5023.2    0.05       0
Bank Sta=5015.2,5023.2
Exp/Cntr=0.3,0.1

Type RM Length L Ch R = 1,42600,257,257,257
BEGIN DESCRIPTION:
Dry Lacy Fork 2351
END DESCRIPTION:
XS GIS Cut Line= 4
      2760632.99      6891276.34      2760166.55      6891635.54
      2759186.75      6891677.46      2758364.64      6891760.40
#Sta/Elev= 30
  3435.7  500.76  3550.8  486.92  3627.7  480.98  3764.7  471.58  3835.8  474.36
  3893.3  473.12  3899.6  471.31  3949.5  469.56  4385.3  469.38  4445.4  468.35
  4545.4  469.31  4625.5  466.64  4665.6  468.06  4705.6  467.23  4733.8  468.56
  4955.8  468.32  4970.9  467.78  4975.9  465.92  5036.0  464.96  5060.7  462.62
  5062.2  462.12  5071.7  462.62  5085.7  466.97  5096.3  468.37  5247.1  467.28
  5397.8  470.13  5428.0  469.69  5491.0  470.82  5699.4  479.15  5831.4  478.39
#Mann=4,-1,0
  3435.7    0.12       0  3627.7    0.05       0  5060.7    0.05       0
  5071.7    0.05       0
Bank Sta=5060.7,5071.7
Exp/Cntr=0.3,0.1

Type RM Length L Ch R = 1,42343,1138,1138,1138
BEGIN DESCRIPTION:
Dry Lacy Fork 2349
END DESCRIPTION:
XS GIS Cut Line= 4
      2760331.26      6891137.37      2759963.33      6891408.21
      2759072.73      6891466.42      2758190.08      6891515.77
#Sta/Elev= 30
  3654.2  500.57  3709.0  499.08  3903.9  482.94  3924.7  479.02  3950.7  479.18
  4109.2  470.77  4281.8  469.19  4381.2  468.67  4480.6  467.25  4679.3  467.25
  4778.7  467.92  4878.0  468.26  4908.6  468.20  4940.2  468.49  4960.2  463.09
  4974.5  462.37  4976.1  461.87  4986.0  462.37  5000.3  464.26  5020.3  463.40
  5030.3  467.00  5040.4  468.24  5348.0  467.21  5360.9  469.08  5390.9  467.78
  5473.8  468.75  5601.2  473.89  5691.4  471.88  5751.5  475.50  5887.6  477.64
#Mann=14,-1,0
  3654.2    0.05       0  3709.0    0.12       0  3950.7    0.05       0
  4281.8    0.12       0  4381.2     0.1       0  4480.6    0.12       0
  4679.3     0.1       0  4778.7    0.12       0  4878.0     0.1       0
  4908.6    0.05       0  4974.5    0.05       0  4986.0    0.05       0
  5348.0    0.12       0  5473.8    0.05       0
Bank Sta=4974.5,4986
Exp/Cntr=0.3,0.1

Type RM Length L Ch R = 1,41205,472,472,472
BEGIN DESCRIPTION:
Dry Lacy Fork 2350
END DESCRIPTION:
XS GIS Cut Line= 3
      2759771.39      6890918.03      2758179.58      6890949.32
      2757759.80      6891348.36
#Sta/Elev= 30
  3454.2  489.77  3459.6  488.62  3509.6  486.34  3529.6  484.62  3649.8  480.31
  3749.6  477.79  3839.7  477.62  3879.7  474.72  3930.7  472.86  3969.7  471.25
  4114.2  469.60  4219.7  470.37  4276.9  469.18  4371.7  467.00  4549.8  465.25
  5009.9  465.66  5029.9  465.15  5039.9  460.82  5041.4  460.32  5051.4  460.82
  5064.3  463.20  5071.2  465.35  5078.5  465.91  5120.6  465.94  5160.5  468.34
  5241.1  471.86  5354.4  475.18  5453.1  476.73  5559.4  475.98  5625.5  477.07
#Mann=8,-1,0
  3454.2    0.12       0  3649.8     0.1       0  3930.7    0.12       0
  4114.2    0.05       0  4276.9    0.12       0  5039.9    0.07       0
  5051.4    0.12       0  5160.5    0.05       0
Bank Sta=5039.9,5051.4
Exp/Cntr=0.3,0.1

Type RM Length L Ch R = 1,40733,410,410,410
BEGIN DESCRIPTION:
Dry Lacy Fork 2352
END DESCRIPTION:
XS GIS Cut Line= 3
      2759190.33      6890611.59      2758082.45      6890631.76
      2757294.46      6891435.58
#Sta/Elev= 30
  3796.6  484.18  3941.0  481.55  4171.0  480.55  4521.0  465.44  4916.8  464.81
  4937.0  465.58  4966.6  460.15  4968.2  459.65  4978.2  460.15  4979.4  461.86
  4993.5  466.15  5007.7  465.33  5014.8  462.47  5029.0  461.70  5071.4  466.26
  5092.5  461.92  5099.7  461.82  5106.7  464.08  5113.7  463.28  5120.8  464.96
  5135.0  465.52  5234.0  468.81  5283.4  468.78  5400.3  471.84  5509.7  469.95
  5672.5  474.43  5806.8  473.87  5827.9  475.05  5863.3  472.38  6030.3  476.67
#Mann=5,-1,0
  3796.6    0.05       0  4916.8    0.12       0  4966.6    0.07       0
  4978.2    0.12       0  5400.3    0.05       0
Bank Sta=4966.6,4978.2
Exp/Cntr=0.3,0.1

Type RM Length L Ch R = 1,40323,535,535,535
BEGIN DESCRIPTION:
Dry Lacy Fork 2353
END DESCRIPTION:
XS GIS Cut Line= 3
      2758602.12      6889694.53      2757788.18      6890382.56
      2757170.39      6891360.13
#Sta/Elev= 30
  3940.7  482.68  4219.5  476.69  4510.7  474.91  4588.7  476.08  4865.3  467.47
  4915.0  463.67  4937.7  460.13  4939.4  459.63  4949.4  460.13  4950.1  462.20
  4957.0  460.32  4964.4  462.77  4971.0  460.66  4978.7  463.74  5012.9  461.08
  5021.1  460.13  5029.6  462.14  5036.4  464.05  5115.3  464.16  5145.8  462.43
  5340.0  464.45  5355.2  462.05  5384.1  464.69  5601.1  468.06  5658.8  471.99
  5674.0  471.92  5680.0  469.84  5725.8  469.38  5852.5  471.24  6162.9  479.77
#Mann=7,-1,0
  3940.7    0.05       0  4937.7    0.04       0  4949.4    0.05       0
  5012.9    0.12       0  5029.6    0.05       0  5384.1    0.12       0
  5852.5    0.05       0
Bank Sta=4937.7,4949.4
Exp/Cntr=0.3,0.1

Type RM Length L Ch R = 1,39788,1455,1455,1455
BEGIN DESCRIPTION:
Dry Lacy Fork 2354
END DESCRIPTION:
XS GIS Cut Line= 3
      2757810.42      6889227.05      2757350.98      6890129.88
      2757068.32      6891247.07
#Sta/Elev= 30
  3982.4  482.58  4159.1  476.19  4309.2  465.02  4368.3  462.76  4403.8  464.88
  4420.5  462.87  4464.9  462.36  4525.4  465.08  4547.8  462.66  4592.7  461.56
  4837.5  461.10  4948.7  462.41  4963.0  460.72  4965.1  458.62  4966.7  458.12
  4976.9  458.62  4995.4  460.97  5034.4  462.11  5110.0  462.59  5182.2  460.19
  5198.4  461.66  5409.2  463.50  5429.8  466.09  5444.5  465.95  5450.4  464.41
  5577.9  468.27  5679.0  470.13  5914.9  475.35  5981.3  476.55  6147.8  480.83
#Mann=7,-1,0
  3982.4    0.05       0  4965.1    0.04       0  4976.9    0.05       0
  5577.9    0.12       0  5679.0    0.05       0  5914.9    0.12       0
  5981.3    0.05       0
Bank Sta=4965.1,4976.9
Exp/Cntr=0.3,0.1

Type RM Length L Ch R = 1,38333,570,570,570
BEGIN DESCRIPTION:
Dry Lacy Fork 2347
END DESCRIPTION:
XS GIS Cut Line= 3
      2756797.88      6887208.70      2756849.11      6889008.86
      2756981.57      6890733.09
#Sta/Elev= 30
  3225.3  483.65  3427.7  474.58  3667.8  468.00  3847.9  460.72  3887.9  460.68
  3907.9  458.40  3927.9  460.80  3947.9  461.18  4338.1  459.82  4391.4  461.20
  4398.1  459.31  4428.1  458.83  4978.3  459.49  4988.3  457.94  4992.4  455.70
  4994.0  455.20  5004.3  455.70  5038.4  459.70  5335.9  459.60  5460.5  460.14
  5710.3  459.96  5761.8  461.85  5870.8  459.77  5931.0  464.10  5958.6  463.81
  6302.1  466.11  6462.6  469.60  6572.9  469.31  6592.9  471.05  6755.5  474.09
#Mann=7,-1,0
  3225.3    0.05       0  4992.4    0.05       0  5004.3    0.05       0
  5335.9    0.12       0  5460.5    0.05       0  5761.8    0.12       0
  5958.6    0.05       0
Bank Sta=4992.4,5004.3
Exp/Cntr=0.3,0.1

Type RM Length L Ch R = 1,37763,814,814,814
BEGIN DESCRIPTION:
Dry Lacy Fork 2346
END DESCRIPTION:
XS GIS Cut Line= 3
      2756537.57      6887280.23      2756582.89      6888585.87
      2756707.44      6890237.65
#Sta/Elev= 30
  3717.4  476.90  3948.3  465.86  4188.5  459.71  4728.8  458.77  4748.8  453.96
  4768.8  458.00  4966.6  459.06  4978.9  457.08  4983.0  452.75  4984.6  452.25
  4994.9  452.75  4998.9  459.18  5019.8  458.94  5109.2  458.67  5119.2  456.07
  5149.3  458.47  5500.3  457.56  5540.4  459.78  5560.5  456.09  5610.6  459.80
  5640.7  454.82  5670.8  460.32  5754.6  459.66  5851.3  459.89  5871.4  457.35
  5944.8  461.20  5988.3  460.16  6129.6  460.92  6571.4  468.22  6680.3  470.35
#Mann=9,-1,0
  3717.4    0.05       0  4983.0    0.04       0  4994.9    0.05       0
  5019.8    0.12       0  5754.6     0.1       0  5944.8    0.12       0
  5988.3     0.1       0  6129.6    0.12       0  6571.4    0.05       0
Bank Sta=4983,4994.9
Exp/Cntr=0.3,0.1

Type RM Length L Ch R = 1,36949,948,948,948
BEGIN DESCRIPTION:
Dry Lacy Fork 2348
END DESCRIPTION:
XS GIS Cut Line= 3
      2756368.57      6886990.43      2755954.51      6888351.07
      2756089.84      6889854.04
#Sta/Elev= 30
  3626.1  482.20  3647.2  480.56  3652.5  481.14  3710.3  476.11  3762.6  473.37
  3783.5  473.64  3822.0  469.71  3887.7  466.31  4138.9  457.58  4308.0  455.68
  4958.4  456.81  4975.1  454.57  4984.4  450.20  4986.4  449.70  4998.0  450.20
  5006.5  453.56  5016.9  454.71  5029.3  459.02  5037.8  459.24  5045.7  457.16
  5078.4  455.52  5389.7  456.67  5520.2  459.23  5610.5  463.31  5640.7  466.76
  5788.0  469.88  5951.9  471.20  6142.7  469.44  6413.8  473.12  6557.4  473.83
#Mann=3,-1,0
  3626.1    0.05       0  4984.4    0.04       0  4998.0    0.05       0
Bank Sta=4984.4,4998
Exp/Cntr=0.3,0.1

Type RM Length L Ch R = 1,36001,714,714,714
BEGIN DESCRIPTION:
Dry Lacy Fork 2344
END DESCRIPTION:
XS GIS Cut Line= 3
      2756057.37      6887119.20      2755135.21      6888132.42
      2754792.87      6889241.14
#Sta/Elev= 30
  3638.4  477.33  3761.2  472.64  3874.1  473.42  3916.7  468.44  3959.2  466.25
  4008.6  461.44  4065.3  460.11  4185.6  454.28  4730.9  455.14  4745.1  454.10
  4766.0  455.52  4857.9  454.49  4928.8  455.96  4993.0  454.31  5004.1  452.37
  5017.4  451.97  5020.6  448.25  5022.6  447.75  5035.2  448.25  5038.3  450.28
  5047.9  452.68  5076.5  454.48  5320.9  455.06  5540.7  460.22  5631.2  461.47
  5663.9  462.55  5669.1  463.52  5804.9  465.99  5832.4  467.95  6168.8  473.33
#Mann=5,-1,0
  3638.4    0.05       0  5020.6    0.04       0  5035.2    0.05       0
  5047.9    0.12       0  5076.5    0.05       0
Bank Sta=5020.6,5035.2
Exp/Cntr=0.3,0.1

Type RM Length L Ch R = 1,35287,804,804,804
BEGIN DESCRIPTION:
Dry Lacy Fork 2345
END DESCRIPTION:
XS GIS Cut Line= 3
      2755302.18      6886846.26      2754800.99      6887548.47
      2753917.18      6888605.03
#Sta/Elev= 30
  4146.8  468.12  4298.8  467.17  4779.2  466.99  4892.5  463.77  4922.0  460.59
  4928.1  458.61  4947.4  458.76  4957.6  459.78  4963.7  457.93  4971.1  448.18
  4973.1  447.68  4985.8  448.18  4997.7  452.06  5008.0  453.91  5086.0  454.61
  5100.3  452.10  5112.4  454.41  5149.7  453.85  5178.4  454.61  5247.3  453.48
  5320.2  454.10  5412.6  453.03  5760.0  454.19  5959.1  458.16  6029.7  461.61
  6094.5  463.28  6121.8  465.11  6300.1  470.81  6335.2  473.21  6387.0  473.46
#Mann=7,-1,0
  4146.8    0.05       0  4947.4     0.1       0  4971.1    0.07       0
  4985.8     0.1       0  4997.7    0.12       0  5112.4     0.1       0
  5247.3    0.05       0
Bank Sta=4971.1,4985.8
Exp/Cntr=0.3,0.1

Type RM Length L Ch R = 1,34483,598,598,598
BEGIN DESCRIPTION:
Dry Lacy Fork 2343
END DESCRIPTION:
XS GIS Cut Line= 3
      2755116.24      6886951.73      2754082.81      6887370.84
      2753605.67      6887826.43
#Sta/Elev= 30
  3889.0  467.43  4170.8  465.40  4219.0  464.43  4248.5  465.48  4272.6  465.02
  4302.1  465.68  4418.0  457.45  4487.0  454.49  4511.1  452.71  4540.5  452.28
  4741.8  451.72  4993.3  452.89  4999.8  451.03  5004.2  451.03  5009.2  446.15
  5015.8  445.75  5017.8  445.25  5030.8  445.75  5037.5  452.06  5044.4  452.66
  5072.7  452.19  5094.1  454.11  5129.3  454.76  5214.2  458.51  5270.8  462.43
  5306.1  462.30  5313.3  463.06  5369.9  464.13  5553.6  465.83  5663.9  468.05
#Mann=3,-1,0
  3889.0    0.05       0  5015.8    0.04       0  5030.8    0.05       0
Bank Sta=5015.8,5030.8
Exp/Cntr=0.3,0.1

Type RM Length L Ch R = 1,33885,136,136,136
BEGIN DESCRIPTION:
Dry Lacy Fork 2342
END DESCRIPTION:
XS GIS Cut Line= 3
      2755059.11      6886947.75      2753822.44      6886946.29
      2752956.28      6887003.22
#Sta/Elev= 30
  3767.0  467.06  3890.1  465.82  4452.9  451.54  4785.3  451.20  4866.9  452.16
  4890.1  452.57  4900.1  449.41  4902.4  444.62  4904.4  444.12  4917.8  444.62
  4950.1  444.72  4970.1  452.01  4980.1  451.44  5010.1  444.95  5020.1  445.66
  5030.2  450.68  5040.2  452.15  5053.7  452.17  5153.6  452.52  5200.5  454.86
  5263.9  459.69  5330.8  464.42  5421.0  466.29  5501.2  465.03  5601.4  465.49
  5791.8  468.19  5801.8  468.59  5811.8  470.33  5831.9  469.20  5871.7  469.34
#Mann=8,-1,0
  3767.0    0.05       0  4452.9    0.12       0  4785.3    0.05       0
  4866.9    0.12       0  4902.4    0.07       0  4917.8    0.12       0
  5053.7    0.05       0  5263.9    0.12       0
Bank Sta=4902.4,4917.8
Exp/Cntr=0.3,0.1

Type RM Length L Ch R = 1,33749,713,713,713
BEGIN DESCRIPTION:
Dry Lacy Fork 2326
END DESCRIPTION:
XS GIS Cut Line= 3
      2754988.24      6886791.45      2753810.51      6886810.48
      2752856.66      6886821.99
#Sta/Elev= 30
  3838.7  466.62  4071.0  464.08  4118.1  464.40  4211.0  462.89  4341.0  457.10
  4468.4  453.28  4611.0  450.90  4844.8  450.70  4951.1  451.48  4961.1  450.54
  4963.4  444.38  4965.4  443.88  4978.8  444.38  4981.1  444.64  4991.1  450.75
  5001.1  451.97  5170.1  451.04  5201.1  450.18  5211.1  451.43  5251.1  452.18
  5261.1  453.78  5431.1  462.78  5470.2  462.31  5475.2  463.15  5551.1  460.63
  5611.1  461.33  5671.0  464.84  5841.2  468.25  5891.2  470.46  5970.5  471.06
#Mann=7,-1,0
  3838.7    0.05       0  4468.4    0.12       0  4844.8     0.1       0
  4963.4    0.07       0  4978.8     0.1       0  5170.1    0.12       0
  5671.0     0.1       0
Bank Sta=4963.4,4978.8
Exp/Cntr=0.3,0.1
