--- Lacy 167.prj (project) ---

Proj Title=Lacy 167 Base Level Engineering
Current Plan=p01
Default Exp/Contr=0.3,0.1
English Units
Geom File=g01
Flow File=f01
Plan File=p01
BEGIN DESCRIPTION:
Lacy 167
END DESCRIPTION:

--- Lacy 167.p01 (plan) ---

Plan Title=Multiple Run
Short Identifier=Multiple
Geom File=g01
Flow File=f01
Subcritical Flow
K Sum by GR= 0
Std Step Tol= 0.01
Critical Tol= 0.01
Num of Std Step Trials= 20
Max Error Tol= 0.3
Flow Tol Ratio= 0.001
Split Flow NTrial= 30
Split Flow Tol= 0.02
Split Flow Ratio= 0.02
Log Output Level= 0
Friction Slope Method= 1
Unsteady Friction Slope Method= 2
Unsteady Bridges Friction Slope Method= 1
Parabolic Critical Depth
Global Vel Dist=  1 , 1 , 1
Global Log Level= 0
CheckData=True
Encroach Param= -1, 0, 0, 0
BEGIN DESCRIPTION:
Multiple Run
END DESCRIPTION:

--- Lacy 167.f01 (steady flow) ---

Flow Title=Multiple
Number of Profiles=7
Profile Names=10-year,25-year,50-year,1pct_min,100-year,1pct_plu,500-year
River Rch & RM= Lacy 167,Reach-1,14906
     248     313     362     208     416     829     547
River Rch & RM= Lacy 167,Reach-1,13247
     445     584     694     410     817    1631    1132
River Rch & RM= Lacy 167,Reach-1,8979
     774    1047    1268     761    1518    3028    2175
River Rch & RM= Lacy 167,Reach-1,2426
     947    1297    1584     958    1912    3814    2785
Boundary for River Rch & Prof#=Lacy 167,Reach-1,1
Up Type=0
Dn Type=3
Dn Slope=0.005
Boundary for River Rch & Prof#=Lacy 167,Reach-1,2
Up Type=0
Dn Type=3
Dn Slope=0.005
Boundary for River Rch & Prof#=Lacy 167,Reach-1,3
Up Type=0
Dn Type=3
Dn Slope=0.005
Boundary for River Rch & Prof#=Lacy 167,Reach-1,4
Up Type=0
Dn Type=3
Dn Slope=0.005
Boundary for River Rch & Prof#=Lacy 167,Reach-1,5
Up Type=0
Dn Type=3
Dn Slope=0.005
Boundary for River Rch & Prof#=Lacy 167,Reach-1,6
Up Type=0
Dn Type=3
Dn Slope=0.005
Boundary for River Rch & Prof#=Lacy 167,Reach-1,7
Up Type=0
Dn Type=3
Dn Slope=0.005

--- Lacy 167.g01 (geometry) ---

Geom Title=Existing Conditions

River Reach=Lacy 167,Reach-1
Reach XY= 30
      2724976.00      6852861.00      2724886.62      6852910.34
      2724669.61      6852803.00      2724589.73      6852574.16
      2724334.50      6852557.53      2723776.00      6852061.00
      2723481.86      6852108.95      2723162.43      6851897.53
      2722779.10      6851309.35      2722868.89      6851161.00
      2722816.83      6851004.01      2722638.96      6850924.63
      2722620.20      6850708.70      2722339.41      6850424.52
      2721755.84      6850561.46      2721424.37      6850314.13
      2721249.10      6850334.98      2721059.77      6849893.79
      2720876.00      6849911.00      2720585.15      6849517.73
      2720546.53      6849130.71      2719884.49      6848857.46
      2719283.80      6848317.21      2719273.74      6847616.94
      2718956.22      6846890.91      2718674.50      6846614.61
      2717476.00      6846261.00      2716799.47      6845434.02
      2716083.81      6844917.19      2716126.00      6844211.00

Type RM Length L Ch R = 1,14906,153,153,153
BEGIN DESCRIPTION:
Lacy 167 578
END DESCRIPTION:
XS GIS Cut Line= 3
      2724967.12      6852678.42      2724910.60      6852911.26
      2724887.71      6853156.59
#Sta/Elev= 30
  4760.4  444.17  4772.2  443.78  4814.5  441.25  4824.2  439.10  4829.3  440.20
  4835.1  437.56  4845.4  437.18  4855.7  437.64  4866.0  436.90  4876.3  437.98
  4896.8  438.09  4912.9  439.16  4943.1  439.09  4959.8  438.37  4979.2  438.10
  4989.4  437.48  4996.4  436.84  4997.1  436.50  4997.4  436.00  5000.9  436.00
  5001.1  436.50  5009.8  436.76  5029.9  438.52  5070.0  439.90  5104.2  440.24
  5200.6  442.77  5213.3  443.65  5220.7  443.25  5230.7  443.48  5246.4  444.34
#Mann=5,-1,0
  4760.4    0.05       0  4772.2     0.1       0  4943.1    0.05       0
  4997.1    0.04       0  5001.1    0.05       0
Bank Sta=4997.1,5001.1
Exp/Cntr=0.3,0.1

Type RM Length L Ch R = 1,14753,156,156,156
BEGIN DESCRIPTION:
Lacy 167 577
END DESCRIPTION:
XS GIS Cut Line= 3
      2724963.60      6852641.91      2724773.80      6852854.93
      2724756.86      6853193.00
#Sta/Elev= 30
  4714.7  445.30  4740.9  443.78  4811.4  440.69  4818.9  438.83  4825.6  439.58
  4833.1  439.07  4839.8  439.50  4847.3  438.62  4854.0  438.74  4868.2  437.67
  4889.1  437.66  4896.6  436.22  4903.3  436.13  4910.9  437.37  4946.0  437.26
  4960.2  436.42  4967.7  436.86  4972.4  435.37  4972.7  434.87  4976.2  434.87
  4976.4  435.37  4981.3  436.67  4996.5  436.60  5036.1  437.52  5046.1  438.52
  5058.6  437.06  5096.2  438.67  5146.3  439.38  5253.6  442.87  5338.5  443.62
#Mann=5,-1,0
  4714.7    0.05       0  4740.9     0.1       0  4972.4    0.05       0
  4976.4     0.1       0  4996.5    0.05       0
Bank Sta=4972.4,4976.4
Exp/Cntr=0.3,0.1

Type RM Length L Ch R = 1,14597,150,150,150
BEGIN DESCRIPTION:
Lacy 167 576
END DESCRIPTION:
XS GIS Cut Line= 3
      2724949.14      6852600.04      2724642.28      6852778.14
      2724619.32      6853140.41
#Sta/Elev= 30
  4645.2  445.67  4655.8  446.03  4661.6  445.11  4680.8  444.68  4736.1  441.67
  4794.9  439.74  4816.5  440.03  4822.3  438.93  4841.0  438.40  4875.2  437.58
  4891.0  437.74  4896.8  437.58  4903.2  436.69  4918.3  437.27  4934.0  436.13
  4957.1  436.20  4984.1  436.06  4992.8  437.00  4995.9  433.56  4996.1  433.06
  4999.6  433.06  4999.9  433.56  5012.9  433.97  5019.0  437.19  5071.1  437.80
  5113.1  438.35  5133.1  440.10  5163.2  438.64  5273.4  441.50  5363.0  442.44
#Mann=7,-1,0
  4645.2    0.05       0  4680.8     0.1       0  4841.0    0.05       0
  4957.1    0.12       0  4995.9    0.07       0  4999.9    0.12       0
  5071.1    0.05       0
Bank Sta=4995.9,4999.9
Exp/Cntr=0.3,0.1

Type RM Length L Ch R = 1,14447,298,298,298
BEGIN DESCRIPTION:
Lacy 167 575
END DESCRIPTION:
XS GIS Cut Line= 3
      2724921.38      6852563.03      2724620.12      6852633.93
      2724131.49      6852804.39
#Sta/Elev= 30
  4695.6  445.77  4729.7  444.28  4803.9  442.16  4838.6  440.46  4896.3  437.66
  4906.6  437.92  4929.5  436.60  4988.8  434.95  5013.1  434.81  5020.0  433.83
  5059.0  434.77  5094.2  435.10  5126.0  433.97  5157.7  434.25  5163.1  433.13
  5166.4  431.84  5166.6  431.34  5170.1  431.34  5170.4  431.84  5178.9  434.03
  5188.9  435.29  5219.9  434.85  5231.9  435.77  5242.5  435.53  5255.8  436.12
  5287.4  436.92  5337.2  436.66  5422.5  436.55  5467.2  437.09  5522.6  437.20
#Mann=9,-1,0
  4695.6    0.05       0  4729.7     0.1       0  4838.6    0.05       0
  5059.0    0.12       0  5166.4    0.05       0  5170.4    0.12       0
  5255.8    0.05       0  5337.2    0.12       0  5467.2    0.05       0
Bank Sta=5166.4,5170.4
Exp/Cntr=0.3,0.1

Type RM Length L Ch R = 1,14149,248,248,248
BEGIN DESCRIPTION:
Lacy 167 573
END DESCRIPTION:
XS GIS Cut Line= 3
      2724889.92      6852398.66      2724390.17      6852576.62
      2723849.56      6852680.58
#Sta/Elev= 30
  4468.2  446.28  4612.5  441.28  4652.8  440.72  4663.4  439.33  4668.8  441.09
  4684.7  441.06  4823.0  435.00  4918.2  433.69  4966.5  433.88  4981.9  431.45
  4997.3  432.95  5023.3  432.59  5033.5  433.31  5043.5  432.68  5094.6  433.51
  5115.7  432.96  5135.3  431.72  5152.4  431.52  5157.5  433.59  5165.9  430.99
  5202.4  430.55  5202.6  430.05  5206.1  430.05  5206.4  430.55  5227.0  433.39
  5237.1  433.71  5288.1  433.03  5309.4  433.69  5451.0  433.30  5549.2  434.42
#Mann=5,-1,0
  4468.2    0.05       0  5115.7    0.12       0  5202.4    0.04       0
  5206.4    0.12       0  5309.4    0.05       0
Bank Sta=5202.4,5206.4
Exp/Cntr=0.3,0.1

Type RM Length L Ch R = 1,13901,115,115,115
BEGIN DESCRIPTION:
Lacy 167 574
END DESCRIPTION:
XS GIS Cut Line= 3
      2724598.79      6852228.18      2724226.66      6852409.15
      2723877.12      6852663.35
#Sta/Elev= 30
  4584.3  444.87  4609.6  445.06  4620.1  441.31  4665.2  439.07  4744.0  436.84
  4754.2  437.53  4766.6  436.44  4901.9  436.40  4932.1  434.68  4954.4  431.71
  4969.5  431.22  4976.6  430.02  4986.5  430.01  4992.1  431.01  5013.6  429.41
  5029.9  430.32  5049.2  431.77  5072.3  431.42  5078.5  431.09  5083.5  427.66
  5083.7  427.16  5087.5  427.66  5093.2  431.47  5164.3  430.84  5179.0  429.97
  5199.9  431.95  5239.9  432.06  5379.9  432.78  5407.0  433.90  5430.3  433.86
#Mann=5,-1,0
  4584.3    0.05       0  5029.9    0.12       0  5083.5    0.04       0
  5087.5    0.12       0  5239.9    0.05       0
Bank Sta=5083.5,5087.5
Exp/Cntr=0.3,0.1

Type RM Length L Ch R = 1,13786,228,228,228
BEGIN DESCRIPTION:
Lacy 167 572
END DESCRIPTION:
XS GIS Cut Line= 3
      2724322.95      6852154.20      2724142.62      6852329.26
      2723830.64      6852685.28
#Sta/Elev= 30
  4749.8  438.39  4830.2  436.19  4872.6  434.05  4957.5  432.55  4964.7  431.06
  4985.8  429.18  4998.8  430.06  5017.6  429.60  5035.3  429.31  5042.9  429.97
  5070.4  429.84  5078.0  430.48  5082.7  426.56  5082.9  426.06  5086.4  426.06
  5086.7  426.56  5098.9  430.34  5113.1  430.93  5120.7  428.38  5127.4  428.82
  5141.6  431.12  5176.7  430.01  5223.8  431.22  5319.1  432.29  5339.9  431.80
  5389.3  432.61  5411.1  434.00  5432.0  433.69  5453.8  434.43  5474.5  434.38
#Mann=5,-1,0
  4749.8    0.05       0  5017.6    0.12       0  5082.7    0.04       0
  5086.7    0.12       0  5223.8    0.05       0
Bank Sta=5082.7,5086.7
Exp/Cntr=0.3,0.1

Type RM Length L Ch R = 1,13558,311,311,311
BEGIN DESCRIPTION:
Lacy 167 571
END DESCRIPTION:
XS GIS Cut Line= 3
      2724220.45      6852014.16      2723944.87      6852212.95
      2723732.93      6852647.75
#Sta/Elev= 30
  4682.9  437.26  4762.4  435.92  4862.1  432.67  4885.3  432.25  4898.0  431.48
  4957.5  430.79  4962.7  429.71  4971.2  428.68  4977.4  428.79  4998.3  426.92
  5004.8  424.29  5005.1  423.79  5008.6  423.79  5008.8  424.29  5013.0  428.14
  5018.9  428.52  5034.4  428.09  5042.8  428.21  5051.3  429.16  5073.9  429.28
  5096.4  428.84  5102.0  428.33  5152.2  428.13  5237.2  428.59  5276.4  429.19
  5310.4  429.86  5349.9  431.98  5378.0  431.90  5454.4  432.63  5506.4  434.39
#Mann=5,-1,0
  4682.9    0.05       0  4957.5    0.12       0  5004.8    0.07       0
  5008.8    0.12       0  5152.2    0.05       0
Bank Sta=5004.8,5008.8
Exp/Cntr=0.3,0.1

Type RM Length L Ch R = 1,13247,227,227,227
BEGIN DESCRIPTION:
Lacy 167 579
END DESCRIPTION:
XS GIS Cut Line= 3
      2723699.38      6851664.30      2723722.49      6852114.25
      2723716.45      6852656.47
#Sta/Elev= 30
  4561.8  433.36  4598.6  432.02  4658.6  430.75  4868.9  427.91  4878.9  426.71
  4888.9  426.48  4898.9  426.34  4919.0  427.85  4939.0  425.28  4949.0  427.70
  4956.5  426.37  4983.7  424.48  4989.1  426.69  4999.1  424.08  5006.2  423.74
  5006.5  423.24  5010.0  423.24  5010.2  423.74  5012.3  423.74  5019.1  426.54
  5059.1  427.39  5126.7  427.21  5249.1  428.05  5339.1  429.31  5399.1  430.95
  5419.1  432.20  5469.1  432.16  5519.1  433.45  5539.1  434.61  5554.6  434.60
#Mann=5,-1,0
  4561.8    0.05       0  4956.5    0.12       0  5006.2    0.07       0
  5010.2    0.12       0  5126.7    0.05       0
Bank Sta=5006.2,5010.2
Exp/Cntr=0.3,0.1

Type RM Length L Ch R = 1,13020,314,314,314
BEGIN DESCRIPTION:
Lacy 167 570
END DESCRIPTION:
XS GIS Cut Line= 3
      2723639.76      6851694.13      2723517.56      6852117.27
      2723473.34      6852507.24
#Sta/Elev= 30
  4565.7  431.53  4598.1  430.36  4614.5  430.18  4636.9  429.27  4704.2  428.14
  4729.0  427.40  4749.8  427.24  4776.6  426.31  4791.4  426.28  4801.8  425.88
  4895.5  425.75  4947.6  426.56  4955.2  424.91  4960.4  424.63  4988.9  425.18
  5010.5  424.89  5018.0  420.01  5018.2  419.51  5021.7  419.51  5022.0  420.01
  5030.0  420.23  5040.1  427.20  5050.1  427.91  5059.8  427.72  5070.3  428.15
  5231.3  429.41  5291.7  430.44  5311.8  431.61  5328.8  431.42  5398.6  432.02
#Mann=3,-1,0
  4565.7    0.05       0  5018.0    0.05       0  5022.0    0.05       0
Bank Sta=5018,5022
Exp/Cntr=0.3,0.1

Type RM Length L Ch R = 1,12706,258,258,258
BEGIN DESCRIPTION:
Lacy 167 569
END DESCRIPTION:
XS GIS Cut Line= 3
      2723575.34      6851622.47      2723259.20      6851955.39
      2723101.82      6852281.60
#Sta/Elev= 30
  4551.4  433.00  4571.1  431.20  4670.2  427.48  4698.6  426.96  4719.6  425.64
  4797.6  424.65  4825.6  423.46  4861.2  422.83  4917.8  423.05  4967.2  424.11
  4981.3  423.17  4983.1  422.33  4993.5  417.16  4993.7  416.66  4997.2  416.66
  4997.5  417.16  5002.7  421.91  5009.2  421.29  5016.7  422.48  5039.0  422.67
  5048.4  422.51  5054.0  421.77  5059.0  422.66  5071.1  424.77  5083.4  425.65
  5116.3  425.58  5167.0  426.91  5189.7  426.25  5234.9  427.76  5372.7  429.36
#Mann=5,-1,0
  4551.4    0.05       0  4983.1    0.12       0  4993.5    0.07       0
  4997.5    0.12       0  5059.0    0.05       0
Bank Sta=4993.5,4997.5
Exp/Cntr=0.3,0.1

Type RM Length L Ch R = 1,12448,236,236,236
BEGIN DESCRIPTION:
Lacy 167 568
END DESCRIPTION:
XS GIS Cut Line= 3
      2723541.98      6851447.64      2723095.86      6851780.14
      2722829.91      6852081.87
#Sta/Elev= 30
  4444.4  433.31  4543.7  429.96  4593.8  429.31  4658.4  426.88  4673.0  425.11
  4679.3  425.76  4693.9  425.19  4723.1  423.03  4823.2  422.38  4837.8  421.09
  4858.6  421.95  4879.4  420.35  4894.0  421.79  4914.9  422.48  4944.1  421.10
  4971.5  421.36  4979.5  421.51  4994.1  420.02  4995.6  416.94  4995.8  416.44
  4999.6  416.94  5008.4  417.62  5015.3  421.86  5070.2  423.95  5128.9  425.90
  5164.0  424.96  5284.5  427.88  5292.0  428.65  5320.5  428.36  5403.0  429.75
#Mann=5,-1,0
  4444.4    0.05       0  4971.5    0.12       0  4995.6    0.07       0
  4999.6    0.12       0  5070.2    0.05       0
Bank Sta=4995.6,4999.6
Exp/Cntr=0.3,0.1

Type RM Length L Ch R = 1,12212,288,288,288
BEGIN DESCRIPTION:
Lacy 167 567
END DESCRIPTION:
XS GIS Cut Line= 3
      2723373.15      6851222.94      2722990.44      6851577.66
      2722731.61      6851813.23
#Sta/Elev= 30
  4481.7  429.77  4513.8  428.22  4591.4  426.16  4613.0  425.11  4662.3  423.93
  4669.1  424.10  4719.0  422.37  4725.8  422.50  4747.3  421.12  4810.9  421.28
  4839.2  420.62  4902.7  420.63  4916.9  420.07  4930.7  420.55  4945.2  419.78
  4973.6  420.42  4987.7  420.30  4993.1  417.11  4993.4  416.61  4996.9  416.61
  4997.1  417.11  5001.9  418.36  5016.1  420.07  5044.5  421.23  5065.4  422.73
  5072.9  423.67  5092.9  423.44  5115.4  423.27  5292.5  426.04  5353.5  426.11
#Mann=5,-1,0
  4481.7    0.05       0  4930.7    0.12       0  4993.1    0.07       0
  4997.1    0.12       0  5092.9    0.05       0
Bank Sta=4993.1,4997.1
Exp/Cntr=0.3,0.1

Type RM Length L Ch R = 1,11924,345,345,345
BEGIN DESCRIPTION:
Lacy 167 565
END DESCRIPTION:
XS GIS Cut Line= 3
      2723353.89      6851012.03      2722812.72      6851357.92
      2722517.27      6851652.39
#Sta/Elev= 30
  4364.5  430.61  4387.0  429.32  4443.5  427.55  4724.3  421.13  4745.5  421.12
  4802.1  419.19  4812.3  419.25  4833.4  417.97  4884.2  418.69  4891.0  419.33
  4927.3  418.53  4969.6  418.64  4978.9  413.48  4982.8  413.40  4983.1  412.90
  4986.6  412.90  4986.8  413.40  4991.0  418.37  4996.2  418.47  5027.8  418.54
  5042.0  419.62  5098.6  420.70  5105.6  421.40  5126.8  421.30  5148.0  423.00
  5190.5  423.77  5254.1  423.95  5261.2  424.88  5339.0  424.26  5423.9  425.21
#Mann=7,-1,0
  4364.5    0.05       0  4387.0    0.12       0  4443.5    0.05       0
  4802.1    0.12       0  4982.8    0.05       0  4986.8    0.12       0
  4996.2    0.05       0
Bank Sta=4982.8,4986.8
Exp/Cntr=0.3,0.1

Type RM Length L Ch R = 1,11579,473,473,473
BEGIN DESCRIPTION:
Lacy 167 566
END DESCRIPTION:
XS GIS Cut Line= 3
      2723253.37      6850882.41      2722799.19      6851087.45
      2722517.02      6851379.62
#Sta/Elev= 30
  4503.8  430.07  4561.2  429.01  4636.1  426.24  4682.3  423.74  4720.4  422.85
  4751.7  421.34  4832.0  419.58  4849.7  418.10  4855.1  418.60  4872.8  417.14
  4884.9  417.64  4899.4  417.18  4939.8  416.57  4976.2  417.27  5021.0  417.01
  5026.1  412.13  5026.4  411.63  5029.9  411.63  5030.1  412.13  5035.1  413.29
  5037.7  414.76  5042.3  417.37  5063.4  416.67  5134.1  418.22  5212.0  421.50
  5226.2  421.20  5233.1  421.79  5303.9  422.68  5367.7  422.32  5408.3  423.78
#Mann=5,-1,0
  4503.8     0.1       0  4899.4    0.12       0  5026.1    0.07       0
  5030.1    0.12       0  5037.7    0.05       0
Bank Sta=5026.1,5030.1
Exp/Cntr=0.3,0.1

Type RM Length L Ch R = 1,11106,274,274,274
BEGIN DESCRIPTION:
Lacy 167 564
END DESCRIPTION:
XS GIS Cut Line= 3
      2722930.71      6850454.06      2722593.33      6850846.27
      2722552.44      6851183.04
#Sta/Elev= 30
  4567.7  425.13  4646.7  422.56  4668.6  422.82  4746.1  420.18  4845.3  417.61
  4880.4  415.60  4930.8  415.13  4937.4  413.92  4945.1  413.86  4951.7  415.06
  4972.6  414.78  4999.1  410.48  4999.3  409.98  5002.8  409.98  5003.1  410.48
  5008.8  411.54  5015.4  415.18  5064.9  415.87  5072.4  410.78  5079.0  415.21
  5084.9  411.28  5099.6  410.66  5104.6  415.22  5110.0  415.65  5120.0  414.77
  5200.6  419.67  5277.7  420.06  5350.0  420.11  5361.8  421.15  5424.3  421.21
#Mann=5,-1,0
  4567.7    0.05       0  4746.1    0.12       0  4999.1    0.07       0
  5003.1    0.12       0  5277.7    0.05       0
Bank Sta=4999.1,5003.1
Exp/Cntr=0.3,0.1

Type RM Length L Ch R = 1,10832,367,367,367
BEGIN DESCRIPTION:
Lacy 167 562
END DESCRIPTION:
XS GIS Cut Line= 3
      2722457.05      6850170.28      2722468.80      6850612.18
      2722433.07      6851011.43
#Sta/Elev= 30
  4570.0  427.88  4630.7  427.23  4651.3  427.45  4710.8  424.24  4717.1  423.34
  4722.1  423.50  4740.8  422.18  4750.8  421.97  4790.8  419.18  4800.8  419.10
  4820.8  417.98  4860.8  416.60  4870.8  415.49  4930.8  412.83  4950.8  413.62
  4970.9  413.01  4990.9  413.56  5000.9  413.39  5007.0  410.52  5007.2  410.02
  5010.7  410.02  5011.0  410.52  5012.1  410.52  5020.9  413.10  5030.9  413.32
  5051.0  414.89  5151.4  415.11  5171.5  417.04  5240.0  417.01  5412.9  418.58
#Mann=5,-1,0
  4570.0    0.05       0  4651.3    0.12       0  5007.0    0.07       0
  5011.0    0.12       0  5240.0    0.05       0
Bank Sta=5007,5011
Exp/Cntr=0.3,0.1

Type RM Length L Ch R = 1,10465,267,267,267
BEGIN DESCRIPTION:
Lacy 167 563
END DESCRIPTION:
XS GIS Cut Line= 3
      2722239.84      6850227.59      2722212.32      6850463.34
      2722181.91      6851013.35
#Sta/Elev= 30
  4765.4  429.41  4784.2  428.08  4809.1  426.60  4838.0  422.57  4843.0  422.69
  4859.4  420.14  4882.5  418.26  4940.0  414.44  4950.1  412.83  4970.2  411.36
  4980.3  409.02  4988.3  408.74  4988.6  408.24  4992.1  408.24  4992.3  408.74
  4999.1  411.45  5010.4  411.49  5031.1  412.72  5078.2  413.23  5100.6  412.88
  5150.6  413.31  5176.7  411.88  5206.8  411.55  5230.8  412.00  5250.8  412.66
  5285.6  414.70  5310.9  417.09  5340.9  416.71  5411.0  417.11  5553.6  418.99
#Mann=8,-1,0
  4765.4    0.05       0  4784.2     0.1       0  4882.5    0.12       0
  4988.3    0.07       0  4992.3    0.12       0  5078.2     0.1       0
  5176.7    0.12       0  5285.6    0.05       0
Bank Sta=4988.3,4992.3
Exp/Cntr=0.3,0.1

Type RM Length L Ch R = 1,10198,298,298,298
BEGIN DESCRIPTION:
Lacy 167 554
END DESCRIPTION:
XS GIS Cut Line= 3
      2722002.29      6850211.64      2721974.38      6850559.12
      2721909.00      6850917.30
#Sta/Elev= 30
  4657.5  427.56  4666.9  427.00  4677.8  425.17  4697.0  423.59  4747.1  417.58
  4784.6  413.88  4800.4  412.50  4827.4  411.48  4877.6  411.40  4917.7  412.17
  4928.1  410.72  4937.8  410.37  4945.8  405.99  4946.0  405.49  4949.5  405.49
  4949.8  405.99  4957.8  410.70  4998.0  409.94  5058.8  410.25  5109.7  411.14
  5130.0  412.26  5140.8  412.11  5180.8  413.70  5211.3  415.60  5221.5  415.57
  5247.3  416.74  5252.4  416.35  5277.7  416.62  5305.6  416.49  5370.2  417.46
#Mann=5,-1,0
  4657.5     0.1       0  4784.6    0.12       0  4945.8    0.07       0
  4949.8    0.12       0  5277.7    0.05       0
Bank Sta=4945.8,4949.8
Exp/Cntr=0.3,0.1

Type RM Length L Ch R = 1,9900,178,178,178
BEGIN DESCRIPTION:
Lacy 167 553
END DESCRIPTION:
XS GIS Cut Line= 3
      2721782.42      6850193.59      2721745.35      6850556.39
      2721705.37      6850854.23
#Sta/Elev= 30
  4631.6  416.78  4649.8  415.42  4729.5  412.38  4749.6  411.06  4820.0  410.08
  4830.0  409.10  4836.7  405.08  4836.9  404.58  4840.4  404.58  4840.7  405.08
  4843.7  408.81  4850.1  405.13  4860.2  409.34  4880.3  409.26  4886.6  408.64
  4890.3  408.27  4910.5  408.58  4930.6  409.94  4943.1  410.19  5001.1  409.82
  5011.0  408.47  5027.6  410.20  5032.6  409.74  5066.5  410.62  5081.7  410.66
  5111.9  412.46  5178.4  413.56  5183.5  413.11  5233.0  413.86  5296.8  415.34
#Mann=5,-1,0
  4631.6    0.05       0  4836.7    0.07       0  4840.7    0.05       0
  4886.6    0.12       0  5066.5    0.05       0
Bank Sta=4836.7,4840.7
Exp/Cntr=0.3,0.1

Type RM Length L Ch R = 1,9722,258,258,258
BEGIN DESCRIPTION:
Lacy 167 552
END DESCRIPTION:
XS GIS Cut Line= 3
      2721696.04      6850118.85      2721602.08      6850464.74
      2721550.85      6850779.47
#Sta/Elev= 30
  4645.4  416.77  4649.1  416.77  4669.1  415.56  4730.5  413.24  4761.6  411.09
  4817.9  409.55  4875.6  409.08  4917.0  408.18  4926.9  409.43  4932.1  408.55
  4937.8  408.73  4971.9  408.22  5007.8  408.37  5020.3  408.71  5030.4  408.73
  5050.7  405.46  5058.8  403.64  5059.1  403.14  5062.6  403.14  5062.8  403.64
  5069.3  406.74  5074.4  406.44  5081.1  408.89  5091.2  410.82  5101.4  411.37
  5182.4  412.19  5212.8  413.06  5243.2  413.50  5320.5  415.29  5322.7  415.03
#Mann=3,-1,0
  4645.4    0.05       0  5058.8    0.05       0  5062.8    0.05       0
Bank Sta=5058.8,5062.8
Exp/Cntr=0.3,0.1

Type RM Length L Ch R = 1,9464,485,485,485
BEGIN DESCRIPTION:
Lacy 167 551
END DESCRIPTION:
XS GIS Cut Line= 3
      2721571.76      6849967.92      2721400.70      6850314.59
      2721351.26      6850640.79
#Sta/Elev= 30
  4617.7  415.50  4690.4  411.38  4707.3  411.29  4712.9  410.65  4729.7  410.42
  4735.3  409.84  4757.8  409.35  4847.6  408.02  4954.3  407.94  4966.8  407.72
  4982.3  406.96  5003.9  406.66  5051.2  407.20  5061.3  407.51  5067.7  408.07
  5091.7  407.32  5101.8  407.35  5111.9  406.71  5131.4  407.40  5136.5  405.26
  5142.2  404.61  5150.4  404.26  5150.6  403.76  5154.1  403.76  5154.4  404.26
  5162.5  408.05  5192.8  410.60  5213.0  411.15  5274.0  411.98  5334.2  413.42
#Mann=3,-1,0
  4617.7    0.05       0  5150.4    0.04       0  5154.4    0.05       0
Bank Sta=5150.4,5154.4
Exp/Cntr=0.3,0.1

Type RM Length L Ch R = 1,8979,286,286,286
BEGIN DESCRIPTION:
Lacy 167 550
END DESCRIPTION:
XS GIS Cut Line= 3
      2721504.64      6849823.45      2721152.39      6850098.41
      2720727.59      6850462.60
#Sta/Elev= 30
  4561.7  415.28  4665.6  408.79  4787.7  406.51  4922.5  405.59  4928.8  403.56
  4934.9  403.30  4935.2  402.80  4938.9  403.30  4957.7  405.83  4972.2  406.09
  4991.9  405.07  5036.2  405.45  5050.4  403.40  5057.0  403.33  5071.3  404.40
  5093.2  403.33  5105.4  404.09  5149.2  406.20  5214.0  405.72  5241.4  406.27
  5298.5  405.64  5306.2  404.63  5348.4  404.60  5376.4  405.70  5390.7  407.75
  5412.1  407.72  5440.1  410.43  5487.7  411.91  5525.7  414.22  5568.1  414.39
#Mann=7,-1,0
  4561.7    0.05       0  4934.9    0.07       0  4938.9    0.05       0
  4991.9    0.12       0  5105.4    0.05       0  5348.4    0.12       0
  5487.7    0.05       0
Bank Sta=4934.9,4938.9
Exp/Cntr=0.3,0.1

Type RM Length L Ch R = 1,8693,237,237,237
BEGIN DESCRIPTION:
Lacy 167 549
END DESCRIPTION:
XS GIS Cut Line= 3
      2721426.47      6849678.78      2721040.70      6849880.22
      2720639.45      6850150.35
#Sta/Elev= 30
  4568.5  413.87  4695.4  407.65  4828.5  405.83  4882.9  405.82  4888.6  405.73
  4894.2  404.59  4896.2  404.18  4910.6  405.95  4918.7  405.76  4927.1  403.62
  4963.9  403.48  4999.0  404.28  5050.7  403.40  5071.7  404.58  5137.7  403.00
  5175.9  402.86  5177.7  402.85  5177.9  402.35  5181.4  402.35  5181.7  402.85
  5266.6  405.23  5287.6  406.20  5296.6  407.39  5317.6  406.93  5383.1  407.87
  5404.6  409.20  5410.6  408.51  5418.0  409.38  5461.6  411.79  5487.4  411.32
#Mann=6,-1,0
  4568.5    0.05       0  4894.2    0.12       0  5175.9    0.05       0
  5177.7    0.07       0  5181.7    0.05       0  5418.0    0.12       0
Bank Sta=5177.7,5181.7
Exp/Cntr=0.3,0.1

Type RM Length L Ch R = 1,8456,249,249,249
BEGIN DESCRIPTION:
Lacy 167 548
END DESCRIPTION:
XS GIS Cut Line= 3
      2721379.91      6849503.63      2720844.74      6849875.66
      2720485.83      6850153.08
#Sta/Elev= 30
  4345.5  412.88  4532.9  407.76  4633.2  406.57  4642.0  405.59  4648.1  406.44
  4669.0  406.43  4690.4  403.50  4698.7  405.12  4719.6  403.67  4727.8  404.96
  4749.3  403.41  4764.2  403.42  4776.5  404.45  4813.1  403.41  4862.8  404.03
  4913.4  402.68  4943.1  403.10  4949.2  402.40  5006.1  401.93  5006.3  401.43
  5010.1  401.93  5067.6  404.32  5099.5  406.46  5172.0  407.95  5185.3  410.01
  5221.8  410.06  5271.6  412.10  5392.0  413.17  5406.5  414.36  5450.9  413.89
#Mann=5,-1,0
  4345.5    0.05       0  4690.4    0.12       0  5006.1    0.07       0
  5010.1    0.12       0  5067.6    0.05       0
Bank Sta=5006.1,5010.1
Exp/Cntr=0.3,0.1

Type RM Length L Ch R = 1,8207,319,319,319
BEGIN DESCRIPTION:
Lacy 167 543
END DESCRIPTION:
XS GIS Cut Line= 3
      2721347.43      6849400.70      2720700.58      6849680.09
      2720420.11      6849908.31
#Sta/Elev= 30
  4292.5  411.59  4360.6  411.81  4431.1  408.33  4501.0  407.17  4544.6  407.54
  4554.1  406.41  4559.5  406.39  4566.4  407.77  4577.3  407.42  4583.0  405.43
  4623.9  405.28  4729.5  403.48  4834.4  404.02  4857.9  402.86  4904.1  402.87
  4955.3  401.41  4955.6  400.91  4959.3  401.41  4974.0  402.02  5036.7  401.94
  5086.3  404.33  5100.6  406.42  5115.0  406.15  5135.8  408.12  5157.7  407.10
  5185.4  409.42  5222.0  409.47  5313.2  412.28  5341.9  411.94  5358.7  413.24
#Mann=5,-1,0
  4292.5    0.05       0  4623.9    0.12       0  4955.3    0.04       0
  4959.3    0.12       0  4974.0    0.05       0
Bank Sta=4955.3,4959.3
Exp/Cntr=0.3,0.1

Type RM Length L Ch R = 1,7888,295,295,295
BEGIN DESCRIPTION:
Lacy 167 544
END DESCRIPTION:
XS GIS Cut Line= 3
      2721344.31      6849282.87      2720553.63      6849430.77
      2720099.34      6849713.54
#Sta/Elev= 30
  4269.7  411.16  4290.1  409.40  4369.7  410.03  4453.0  407.51  4491.8  407.36
  4500.6  406.01  4505.7  406.91  4512.1  404.45  4563.4  405.19  4766.5  402.38
  4919.1  402.06  4980.1  399.34  4994.6  399.89  5000.5  398.84  5008.6  394.85
  5008.9  394.35  5012.6  394.85  5020.8  395.51  5031.0  401.29  5086.5  402.91
  5159.7  403.35  5189.1  404.60  5211.6  404.06  5275.3  406.35  5412.9  406.58
  5436.4  407.22  5442.9  408.49  5500.8  408.28  5537.4  410.48  5609.2  410.72
#Mann=3,-1,0
  4269.7    0.05       0  5008.6    0.04       0  5012.6    0.05       0
Bank Sta=5008.6,5012.6
Exp/Cntr=0.3,0.1

Type RM Length L Ch R = 1,7593,409,409,409
BEGIN DESCRIPTION:
Lacy 167 545
END DESCRIPTION:
XS GIS Cut Line= 3
      2721040.35      6848835.96      2720557.37      6849143.38
      2720074.45      6849700.23
#Sta/Elev= 30
  4427.9  416.14  4456.8  414.68  4515.6  413.89  4527.9  412.49  4563.9  410.85
  4587.2  410.88  4682.0  405.67  4709.5  405.85  4788.7  403.56  4812.4  401.16
  4847.9  399.65  4949.1  398.74  4955.0  397.37  4989.4  394.69  4989.6  394.19
  4993.4  394.69  5000.4  394.73  5027.9  398.92  5049.8  399.97  5120.0  399.55
  5162.7  400.83  5169.4  400.12  5205.5  402.06  5240.6  402.08  5248.2  403.34
  5367.9  404.18  5404.0  406.17  5418.2  405.57  5580.6  409.09  5737.5  411.19
#Mann=3,-1,0
  4427.9    0.05       0  4989.4    0.05       0  4993.4    0.05       0
Bank Sta=4989.4,4993.4
Exp/Cntr=0.3,0.1

Type RM Length L Ch R = 1,7184,268,268,268
BEGIN DESCRIPTION:
Lacy 167 546
END DESCRIPTION:
XS GIS Cut Line= 3
      2720337.21      6848504.43      2720192.97      6849024.10
      2720041.49      6849602.48
#Sta/Elev= 30
  4474.3  412.00  4507.3  408.75  4610.3  403.07  4636.8  402.66  4657.5  400.93
  4699.1  399.97  4718.2  400.14  4750.9  397.90  4870.8  395.14  4896.2  395.74
  4968.9  395.58  4989.6  396.33  5000.0  395.59  5007.4  392.72  5007.7  392.22
  5011.2  392.22  5011.4  392.72  5013.6  392.72  5018.5  395.99  5023.6  397.12
  5051.8  398.02  5058.9  399.23  5093.1  399.01  5104.5  399.28  5113.8  400.83
  5124.1  401.18  5186.1  401.59  5351.5  405.32  5412.2  407.95  5611.5  410.94
#Mann=4,-1,0
  4474.3    0.12       0  4507.3    0.05       0  5007.4    0.04       0
  5011.4    0.05       0
Bank Sta=5007.4,5011.4
Exp/Cntr=0.3,0.1

Type RM Length L Ch R = 1,6916,357,357,357
BEGIN DESCRIPTION:
Lacy 167 547
END DESCRIPTION:
XS GIS Cut Line= 3
      2720236.05      6848432.85      2719966.71      6848901.09
      2719805.38      6849524.27
#Sta/Elev= 30
  4462.2  411.29  4465.9  411.01  4576.9  403.26  4657.4  399.70  4769.5  396.47
  4834.2  395.75  4944.6  394.77  4989.4  396.20  4999.4  394.07  5019.5  392.38
  5019.7  391.88  5023.5  392.38  5033.3  395.64  5136.6  397.71  5148.5  398.65
  5157.2  398.11  5177.9  399.32  5198.5  399.01  5224.5  401.01  5346.3  401.32
  5374.1  402.36  5394.8  404.88  5446.5  404.86  5468.2  406.82  5487.8  406.29
  5539.1  408.51  5584.8  408.41  5611.7  409.49  5625.5  408.60  5646.1  409.11
#Mann=4,-1,0
  4462.2    0.12       0  4465.9    0.05       0  5019.5    0.04       0
  5023.5    0.05       0
Bank Sta=5019.5,5023.5
Exp/Cntr=0.3,0.1

Type RM Length L Ch R = 1,6559,495,495,495
BEGIN DESCRIPTION:
Lacy 167 535
END DESCRIPTION:
XS GIS Cut Line= 3
      2720139.61      6848285.13      2719701.27      6848694.05
      2719384.38      6849060.73
#Sta/Elev= 30
  4406.3  411.83  4414.4  410.75  4505.2  406.00  4519.3  404.22  4540.3  403.67
  4582.8  400.40  4696.2  398.01  4710.3  398.68  4752.8  397.89  4759.7  396.16
  4788.0  393.52  4816.4  394.26  4915.5  394.06  4943.9  395.19  4958.8  394.50
  4971.9  394.55  4983.8  392.23  4984.1  391.73  4987.9  392.23  4993.2  393.61
  5014.0  394.76  5099.4  394.24  5134.5  395.93  5184.9  396.29  5220.0  398.20
  5277.1  399.06  5305.6  401.02  5447.1  405.57  5475.6  403.46  5490.4  403.47
#Mann=6,-1,0
  4406.3    0.12       0  4414.4    0.05       0  4958.8    0.12       0
  4983.8    0.07       0  4987.9    0.12       0  5014.0    0.05       0
Bank Sta=4983.8,4987.9
Exp/Cntr=0.3,0.1

Type RM Length L Ch R = 1,6064,453,453,453
BEGIN DESCRIPTION:
Lacy 167 534
END DESCRIPTION:
XS GIS Cut Line= 3
      2719922.44      6848023.78      2719390.25      6848298.92
      2719020.51      6848809.26
#Sta/Elev= 30
  4311.8  411.86  4330.3  408.76  4409.2  404.84  4442.3  401.73  4470.0  401.54
  4508.7  399.34  4589.2  397.59  4641.6  395.19  4708.0  393.98  4724.3  394.79
  4790.6  391.60  4950.1  391.86  5015.2  392.44  5027.7  391.07  5028.1  390.57
  5032.1  391.07  5044.6  391.49  5050.7  393.51  5065.4  394.90  5086.3  394.87
  5115.7  396.59  5130.4  396.16  5209.8  398.67  5222.4  400.08  5237.1  399.62
  5337.6  403.42  5358.5  403.26  5395.1  405.26  5488.4  406.30  5541.1  405.54
#Mann=5,-1,0
  4311.8    0.05       0  4790.6    0.12       0  4950.1    0.05       0
  5027.7    0.04       0  5032.1    0.05       0
Bank Sta=5027.7,5032.1
Exp/Cntr=0.3,0.1

Type RM Length L Ch R = 1,5611,328,328,328
BEGIN DESCRIPTION:
Lacy 167 533
END DESCRIPTION:
XS GIS Cut Line= 3
      2719923.76      6847964.94      2719327.66      6847958.05
      2718781.22      6847962.71
#Sta/Elev= 30
  4402.5  412.52  4460.3  408.75  4610.3  402.03  4620.3  400.79  4630.3  398.66
  4640.3  397.86  4660.3  398.42  4710.3  395.31  4730.3  393.21  4770.3  391.82
  4787.3  391.98  4840.3  391.84  4858.1  390.95  4858.5  390.45  4862.1  390.45
  4862.5  390.95  4893.3  391.22  4930.3  392.06  4940.3  390.96  5010.3  391.37
  5040.3  390.96  5048.5  391.48  5150.3  392.82  5191.7  395.05  5210.3  396.50
  5230.3  396.47  5250.3  397.58  5370.3  398.56  5430.3  400.81  5545.1  401.81
#Mann=7,-1,0
  4402.5    0.05       0  4787.3    0.12       0  4858.1    0.04       0
  4862.5    0.12       0  4893.3    0.05       0  5048.5    0.12       0
  5191.7    0.05       0
Bank Sta=4858.1,4862.5
Exp/Cntr=0.3,0.1

Type RM Length L Ch R = 1,5283,166,166,166
BEGIN DESCRIPTION:
Lacy 167 532
END DESCRIPTION:
XS GIS Cut Line= 3
      2719872.33      6847652.03      2719276.16      6847645.14
      2718726.26      6847670.50
#Sta/Elev= 30
  4404.0  417.73  4424.4  416.63  4460.3  414.47  4523.3  409.49  4580.3  404.42
  4600.3  403.18  4610.3  403.12  4620.3  402.45  4630.3  401.20  4640.4  400.63
  4650.4  400.65  4680.4  398.33  4720.4  396.72  4790.4  392.70  4810.4  392.40
  4830.4  391.10  4878.1  390.84  4878.6  390.34  4882.2  390.34  4882.6  390.84
  5170.6  391.13  5190.6  391.52  5270.7  395.69  5340.7  398.13  5350.7  399.15
  5420.8  401.16  5440.8  401.36  5454.4  402.30  5470.9  401.90  5550.7  402.18
#Mann=5,-1,0
  4404.0    0.05       0  4424.4    0.12       0  4523.3    0.05       0
  4878.1    0.03       0  4882.6    0.05       0
Bank Sta=4878.1,4882.6
Exp/Cntr=0.3,0.1

Type RM Length L Ch R = 1,5117,343,343,343
BEGIN DESCRIPTION:
Lacy 167 530
END DESCRIPTION:
XS GIS Cut Line= 3
      2719809.07      6847466.99      2719232.63      6847495.20
      2718680.67      6847496.26
#Sta/Elev= 30
  4416.5  409.39  4420.6  409.39  4429.6  408.51  4439.6  406.79  4449.6  406.05
  4459.6  406.01  4499.7  403.17  4509.7  403.05  4539.7  401.57  4549.7  400.71
  4579.8  399.71  4619.8  397.02  4679.9  395.56  4699.9  394.75  4729.9  392.35
  4767.7  391.05  4768.2  390.55  4771.8  390.55  4772.2  391.05  5180.3  391.34
  5190.3  392.14  5210.3  392.42  5250.3  394.14  5290.3  395.22  5380.3  398.91
  5430.3  399.37  5440.3  399.12  5470.3  399.93  5510.3  399.76  5545.6  400.20
#Mann=3,-1,0
  4416.5    0.05       0  4767.7    0.03       0  4772.2    0.05       0
Bank Sta=4767.7,4772.2
Exp/Cntr=0.3,0.1

Type RM Length L Ch R = 1,4774,696,696,696
BEGIN DESCRIPTION:
Lacy 167 531
END DESCRIPTION:
XS GIS Cut Line= 3
      2719868.77      6847042.37      2719077.97      6847197.21
      2718651.48      6847474.82
#Sta/Elev= 30
  4193.9  413.12  4212.4  411.68  4217.5  412.01  4227.3  411.51  4247.7  409.71
  4263.9  407.64  4298.6  405.93  4329.2  403.24  4423.5  400.26  4431.1  399.09
  4451.5  397.76  4469.9  397.11  4475.0  397.39  4543.2  394.69  4578.0  392.18
  4604.3  391.16  4781.7  391.09  4782.1  390.59  4785.7  390.59  4786.2  391.09
  4869.3  391.89  4950.8  391.90  4989.9  391.35  5214.2  391.67  5220.1  392.90
  5228.8  393.36  5300.4  395.67  5488.9  399.63  5494.8  400.26  5508.6  399.91
#Mann=3,-1,0
  4193.9    0.05       0  4781.7    0.03       0  4786.2    0.05       0
Bank Sta=4781.7,4786.2
Exp/Cntr=0.3,0.1

Type RM Length L Ch R = 1,4078,156,156,156
BEGIN DESCRIPTION:
Lacy 167 529
END DESCRIPTION:
XS GIS Cut Line= 4
      2719470.18      6846283.74      2718990.12      6846183.51
      2718684.68      6846675.50      2718626.80      6847526.13
#Sta/Elev= 30
  3971.5  402.55  4010.4  402.11  4037.1  403.22  4047.3  402.77  4060.4  400.17
  4077.9  399.40  4155.3  398.92  4205.3  400.06  4241.4  399.15  4255.3  399.63
  4355.4  398.02  4400.2  396.17  4450.3  395.69  4461.5  394.92  4529.6  393.89
  4551.1  392.92  4572.4  390.81  4941.5  391.25  5044.2  390.79  5044.7  390.29
  5048.4  390.29  5048.8  390.79  5098.4  391.40  5116.7  390.90  5377.3  391.34
  5517.6  395.05  5547.7  396.44  5748.1  398.69  5798.2  398.70  5893.6  400.84
#Mann=3,-1,0
  3971.5    0.05       0  5044.2    0.03       0  5048.8    0.05       0
Bank Sta=5044.2,5048.8
Exp/Cntr=0.3,0.1

Type RM Length L Ch R = 1,3922,100,100,100
BEGIN DESCRIPTION:
Lacy 167 3411
END DESCRIPTION:
XS GIS Cut Line= 6
      2719474.52      6846192.12      2719219.95      6846049.93
      2719026.44      6845958.96      2718633.43      6846036.35
      2718562.99      6846102.86      2718564.88      6847556.70
#Sta/Elev= 30
  3502.9  401.81  3532.9  404.39  3592.3  401.24  3673.0  401.27  3695.1  404.54
  3738.5  404.34  3753.2  402.26  3776.1  404.53  3849.7  402.90  3855.2  404.47
  3895.3  401.25  3900.8  403.44  3915.8  400.91  3916.2  400.41  3920.4  400.91
  3923.6  403.92  3940.9  401.65  3946.4  403.82  3963.7  402.39  3969.2  404.09
  4110.7  404.89  4365.5  404.68  4404.1  402.76  4408.0  404.68  4474.1  404.72
  4481.1  402.96  4488.0  404.62  4495.2  402.19  4543.9  405.05  5959.6  403.74
#Mann=3,-1,0
  3502.9    0.05       0  3915.8    0.05       0  3920.4    0.05       0
Bank Sta=3915.8,3920.4
Exp/Cntr=0.3,0.1

Type RM Length L Ch R = 1,3822,190,190,190
BEGIN DESCRIPTION:
Lacy 167 527
END DESCRIPTION:
XS GIS Cut Line= 3
      2718497.13      6845767.18      2718475.69      6846566.76
      2718483.66      6847491.76
#Sta/Elev= 30
  4205.9  396.78  4289.8  396.93  4299.8  396.19  4329.8  396.25  4409.8  394.23
  4489.8  390.87  4499.8  389.86  4529.8  388.85  4589.9  385.30  4639.9  383.56
  4870.0  380.84  4920.0  381.12  4930.0  380.11  4980.0  380.78  5037.7  379.98
  5038.2  379.48  5041.9  379.48  5042.4  379.98  5070.0  381.14  5080.0  380.47
  5120.0  380.86  5210.0  382.97  5260.0  385.99  5300.0  387.43  5370.0  391.24
  5460.0  394.98  5520.0  396.13  5550.0  397.73  5780.0  401.20  5930.8  401.84
#Mann=3,-1,0
  4205.9    0.05       0  5037.7    0.05       0  5042.4    0.05       0
Bank Sta=5037.7,5042.4
Exp/Cntr=0.3,0.1

Type RM Length L Ch R = 1,3632,295,295,295
BEGIN DESCRIPTION:
Lacy 167 528
END DESCRIPTION:
XS GIS Cut Line= 3
      2718302.87      6845783.45      2718300.65      6846514.22
      2718296.06      6847220.63
#Sta/Elev= 30
  4273.8  397.23  4351.4  397.71  4381.4  395.16  4421.4  394.00  4431.4  394.60
  4471.4  391.24  4501.4  391.24  4521.4  388.61  4551.4  387.22  4581.4  387.30
  4591.4  386.05  4641.4  384.12  4801.4  381.15  4871.4  378.87  4961.4  379.34
  4971.4  378.40  4981.4  372.92  4989.0  372.46  4989.5  371.96  4993.7  372.46
  5000.5  377.34  5004.6  377.34  5011.4  379.50  5051.4  379.74  5061.4  378.05
  5111.4  378.65  5171.4  383.09  5211.4  384.93  5541.4  398.28  5711.0  400.59
#Mann=3,-1,0
  4273.8    0.05       0  4989.0    0.04       0  4993.7    0.05       0
Bank Sta=4989,4993.7
Exp/Cntr=0.3,0.1

Type RM Length L Ch R = 1,3337,361,361,361
BEGIN DESCRIPTION:
Lacy 167 512
END DESCRIPTION:
XS GIS Cut Line= 3
      2718163.28      6845819.14      2718034.72      6846424.03
      2717937.28      6847027.82
#Sta/Elev= 30
  4394.3  395.33  4437.1  394.71  4518.9  389.41  4552.1  389.61  4559.8  387.68
  4570.0  386.94  4621.1  385.56  4631.3  383.96  4651.8  382.93  4690.7  381.80
  4702.9  382.15  4723.3  380.36  4846.0  378.33  4876.7  376.87  4958.5  377.14
  4983.3  378.06  4986.8  373.81  4987.3  373.31  4991.5  373.81  4999.4  374.17
  5008.6  378.21  5080.5  377.42  5097.3  379.87  5102.3  379.26  5121.1  381.06
  5202.1  383.98  5273.0  385.51  5293.3  386.76  5384.4  388.71  5624.3  397.56
#Mann=3,-1,0
  4394.3    0.05       0  4986.8    0.04       0  4991.5    0.05       0
Bank Sta=4986.8,4991.5
Exp/Cntr=0.3,0.1

Type RM Length L Ch R = 1,2976,550,550,550
BEGIN DESCRIPTION:
Lacy 167 511
END DESCRIPTION:
XS GIS Cut Line= 3
      2717907.23      6845839.24      2717702.18      6846322.82
      2717667.37      6846876.97
#Sta/Elev= 30
  4486.9  392.45  4521.4  390.90  4527.7  389.02  4543.1  388.14  4575.0  387.64
  4586.6  385.84  4604.1  384.76  4619.2  384.20  4627.8  384.96  4640.9  383.06
  4680.5  379.91  4704.2  380.81  4762.4  376.93  4803.8  375.93  4857.1  376.70
  4886.2  375.95  4962.6  377.22  4977.6  376.66  4989.3  374.28  4989.9  373.78
  4994.1  374.28  5008.5  377.28  5040.4  376.76  5230.8  379.68  5270.9  382.07
  5341.0  383.60  5361.0  385.55  5421.1  386.22  5507.9  390.32  5567.4  391.41
#Mann=3,-1,0
  4486.9    0.05       0  4989.3    0.04       0  4994.1    0.05       0
Bank Sta=4989.3,4994.1
Exp/Cntr=0.3,0.1

Type RM Length L Ch R = 1,2426,314,314,314
BEGIN DESCRIPTION:
Lacy 167 46
END DESCRIPTION:
XS GIS Cut Line= 3
      2717575.99      6845611.01      2717326.00      6846011.00
      2716626.03      6846610.97
#Sta/Elev= 30
  4522.1  391.01  4608.8  386.95  4624.1  383.63  4630.0  385.22  4645.3  383.00
  4660.6  376.58  4667.9  376.86  4724.3  374.39  4818.7  376.08  4833.5  375.55
  4891.8  374.82  4964.9  376.15  4977.6  372.24  4978.3  371.74  4982.8  372.24
  5000.9  372.51  5007.5  374.57  5320.3  376.03  5348.8  377.37  5419.1  377.22
  5482.7  380.00  5539.8  380.11  5603.5  383.18  5652.9  383.74  5681.4  386.27
  5724.2  386.61  5759.3  389.62  5787.9  389.62  5880.1  392.81  5915.7  395.47
#Mann=5,-1,0
  4522.1    0.05       0  4667.9    0.12       0  4833.5    0.05       0
  4977.6    0.04       0  4982.8    0.05       0
Bank Sta=4977.6,4982.8
Exp/Cntr=0.3,0.1

Type RM Length L Ch R = 1,2112,340,340,340
BEGIN DESCRIPTION:
Lacy 167 510
END DESCRIPTION:
XS GIS Cut Line= 3
      2717528.71      6845440.79      2717133.20      6845774.56
      2716482.73      6846466.08
#Sta/Elev= 30
  4486.8  394.01  4516.7  394.32  4559.6  391.95  4581.7  391.67  4772.1  380.81
  4793.7  379.40  4815.7  375.75  4836.6  374.29  4900.3  373.27  4971.8  374.53
  4978.3  372.98  4985.5  373.03  4990.0  372.69  4990.7  372.19  4995.2  372.69
  4999.2  374.46  5006.9  374.61  5063.6  373.04  5120.2  374.27  5374.7  374.33
  5410.3  376.06  5502.2  377.43  5523.2  379.23  5579.8  379.61  5615.5  382.08
  5629.6  381.51  5693.1  385.12  5700.0  384.30  5735.6  387.04  5953.7  394.14
#Mann=5,-1,0
  4486.8    0.05       0  4772.1    0.12       0  4985.5    0.05       0
  4990.0    0.05       0  4995.2    0.05       0
Bank Sta=4990,4995.2
Exp/Cntr=0.3,0.1

Type RM Length L Ch R = 1,1772,365,365,365
BEGIN DESCRIPTION:
Lacy 167 509
END DESCRIPTION:
XS GIS Cut Line= 3
      2717211.00      6845267.24      2716896.50      6845530.11
      2716282.69      6846160.15
#Sta/Elev= 30
  4589.3  389.75  4666.4  387.34  4738.0  383.77  4758.8  381.54  4872.0  375.23
  4894.1  374.80  4908.5  373.06  4943.6  373.37  4950.1  374.42  4957.9  373.82
  4964.4  374.84  4986.5  374.51  4993.1  372.25  4996.3  373.47  5007.2  374.28
  5021.4  372.21  5028.4  374.25  5035.5  373.57  5056.7  374.33  5085.0  373.36
  5099.1  371.68  5181.4  371.18  5182.1  370.68  5186.6  371.18  5304.3  373.83
  5339.6  372.27  5360.9  373.91  5728.5  386.22  5855.8  388.73  5878.8  388.34
#Mann=3,-1,0
  4589.3    0.05       0  5181.4    0.04       0  5186.6    0.05       0
Bank Sta=5181.4,5186.6
Exp/Cntr=0.3,0.1

Type RM Length L Ch R = 1,1407,167,167,167
BEGIN DESCRIPTION:
Lacy 167 508
END DESCRIPTION:
XS GIS Cut Line= 3
      2717007.66      6845106.65      2716597.41      6845315.39
      2716128.58      6845964.36
#Sta/Elev= 30
  4564.0  386.92  4628.1  384.16  4650.4  382.17  4656.0  380.59  4672.6  379.78
  4678.2  381.16  4689.3  380.76  4845.0  372.74  4961.8  370.66  5000.7  372.39
  5006.3  367.02  5012.0  366.31  5012.8  365.81  5017.3  366.31  5022.3  369.29
  5048.1  371.19  5116.0  371.12  5122.2  371.87  5136.9  370.73  5252.2  370.69
  5260.1  371.56  5288.1  371.20  5358.9  372.34  5415.4  374.70  5430.1  376.24
  5524.5  379.96  5643.8  387.69  5681.5  390.02  5717.1  390.89  5824.9  389.97
#Mann=7,-1,0
  4564.0    0.05       0  5012.0    0.04       0  5017.3    0.05       0
  5048.1    0.12       0  5260.1    0.05       0  5288.1     0.1       0
  5643.8    0.05       0
Bank Sta=5012,5017.3
Exp/Cntr=0.3,0.1

Type RM Length L Ch R = 1,1240,385,385,385
BEGIN DESCRIPTION:
Lacy 167 507
END DESCRIPTION:
XS GIS Cut Line= 3
      2716891.81      6844968.92      2716480.65      6845219.18
      2715992.57      6845617.15
#Sta/Elev= 30
  4521.1  380.44  4555.6  379.24  4571.0  377.20  4592.4  376.18  4745.4  371.81
  4797.2  372.05  4809.3  371.15  4919.7  370.37  4972.0  370.90  4984.5  372.65
  4993.3  369.01  4996.5  366.70  4997.3  366.20  5001.8  366.70  5002.2  369.23
  5028.4  370.85  5061.4  370.72  5178.8  370.75  5199.3  370.02  5213.7  371.36
  5241.0  370.71  5294.5  371.68  5309.0  372.71  5383.1  376.78  5440.6  378.18
  5454.9  379.57  5547.6  383.45  5568.4  383.44  5582.8  385.02  5632.2  386.17
#Mann=7,-1,0
  4521.1    0.05       0  4996.5    0.04       0  5001.8    0.05       0
  5061.4    0.12       0  5178.8    0.05       0  5294.5     0.1       0
  5309.0    0.12       0
Bank Sta=4996.5,5001.8
Exp/Cntr=0.3,0.1

Type RM Length L Ch R = 1,855,572,572,572
BEGIN DESCRIPTION:
Mapping XS 806a11ab
END DESCRIPTION:
XS GIS Cut Line= 3
      2716859.01      6844928.16      2716296.10      6844902.94
      2715844.58      6845295.98
#Sta/Elev= 30
  4275.7  376.87  4348.8  373.30  4478.9  370.61  4819.3  370.48  4841.5  369.17
  4873.4  370.41  4979.7  370.46  4994.0  372.18  5008.2  369.61  5014.8  366.33
  5019.7  366.03  5020.5  365.53  5025.1  366.03  5029.1  368.52  5036.7  370.24
  5053.1  370.47  5119.9  369.47  5128.8  368.09  5157.3  369.62  5163.9  369.03
  5192.4  371.89  5206.6  374.94  5220.9  376.41  5256.0  378.21  5276.9  380.55
  5333.8  383.69  5341.5  382.79  5355.7  384.77  5397.5  387.51  5437.8  388.06
#Mann=5,-1,0
  4275.7    0.05       0  5019.7    0.04       0  5025.1    0.05       0
  5053.1     0.1       0  5119.9    0.05       0
Bank Sta=5019.7,5025.1
Exp/Cntr=0.3,0.1

Type RM Length L Ch R = 1,283,0,0,0
BEGIN DESCRIPTION:
Lacy 167 506
END DESCRIPTION:
XS GIS Cut Line= 4
      2716853.24      6844921.24      2716239.93      6844474.08
      2716001.73      6844476.34      2715831.47      6845286.63
#Sta/Elev= 30
  4076.9  376.56  4183.2  371.31  4239.6  370.18  4354.7  369.62  4505.3  370.16
  4733.2  368.84  4879.8  368.95  4889.8  369.85  4919.8  368.79  4969.8  368.71
  4989.8  365.80  5019.8  369.44  5036.5  365.85  5041.5  366.05  5049.8  364.56
  5167.6  364.49  5168.4  363.99  5173.1  364.49  5175.4  365.98  5181.1  366.66
  5293.5  366.74  5364.7  367.90  5477.4  366.76  5608.9  370.91  5661.5  375.10
  5663.7  375.21  5692.0  377.43  5743.1  379.09  5803.2  383.34  5902.1  387.26
#Mann=5,-1,0
  4076.9    0.05       0  5167.6    0.05       0  5173.1    0.05       0
  5661.5     0.1       0  5663.7    0.05       0
Bank Sta=5167.6,5173.1
Exp/Cntr=0.3,0.1

Chan Stop Cuts=-1
