HEC-RAS study Mill Creek.prj: Mill Creek Base Level Engineering

--- Mill Creek.g01 (geometry) --- (continued)

Type RM Length L Ch R = 1,25714,270,270,270
BEGIN DESCRIPTION:
Mill Creek25713.76
END DESCRIPTION:
XS GIS Cut Line= 3
      2754824.54      6819659.94      2754854.03      6820413.98
      2754862.01      6820994.31
#Sta/Elev= 30
  4248.4  439.81  4299.5  436.97  4379.6  430.89  4414.2  431.16  4469.6  428.79
  4569.7  429.91  4667.2  427.93  4729.8  427.43  4769.9  424.19  4799.9  426.18
  4910.0  426.40  4970.0  427.39  4980.0  427.19  4990.0  424.50  4994.3  421.27
  4994.8  420.77  5003.2  420.77  5003.7  421.27  5010.0  424.06  5020.0  426.24
  5030.0  427.22  5120.1  427.91  5170.1  427.45  5180.1  426.51  5220.1  427.07
  5260.1  428.83  5380.1  437.40  5440.1  440.14  5480.1  442.94  5583.4  446.01
#Mann=3,-1,0
  4248.4    0.05       0  4994.3    0.05       0  5003.7    0.05       0
Bank Sta=4994.3,5003.7
Exp/Cntr=0.3,0.1

Type RM Length L Ch R = 1,25444,337,337,337
BEGIN DESCRIPTION:
Mill Creek25443.89
END DESCRIPTION:
XS GIS Cut Line= 3
      2754533.85      6819694.51      2754584.15      6820409.23
      2754625.88      6820870.86
#Sta/Elev= 30
  4283.3  433.85  4329.9  430.74  4390.1  428.28  4500.3  426.66  4650.7  426.01
  4680.8  424.84  4730.9  425.49  4750.9  423.53  4761.0  423.43  4781.0  425.27
  4841.2  424.90  4901.3  425.41  4961.5  426.89  4981.5  423.38  4991.5  423.24
  4993.5  420.42  4994.0  419.92  5002.4  419.92  5002.9  420.42  5011.6  420.58
  5021.6  426.81  5122.1  425.03  5182.1  424.95  5192.3  424.54  5232.5  424.97
  5262.6  426.64  5322.9  430.98  5353.0  433.73  5363.0  435.21  5463.3  440.09
#Mann=3,-1,0
  4283.3    0.05       0  4993.5    0.05       0  5002.9    0.05       0
Bank Sta=4993.5,5002.9
Exp/Cntr=0.3,0.1

Type RM Length L Ch R = 1,25107,180,180,180
BEGIN DESCRIPTION:
Mill Creek25107.06
END DESCRIPTION:
XS GIS Cut Line= 3
      2754197.28      6819752.19      2754321.04      6820226.21
      2754544.04      6820851.63
#Sta/Elev= 30
  4516.3  436.84  4577.1  433.16  4652.2  430.27  4836.0  425.65  4918.1  424.26
  4925.1  423.63  4930.3  418.44  4938.8  420.51  4949.2  418.27  4959.5  417.61
  4965.6  417.61  4970.7  423.35  4980.2  422.98  4985.6  417.23  4986.1  416.73
  4995.3  417.23  5000.8  417.69  5006.0  422.04  5011.4  420.98  5021.9  425.16
  5031.6  425.50  5036.9  422.86  5043.1  424.92  5082.3  425.03  5255.5  425.17
  5452.3  423.66  5483.1  424.55  5544.7  428.95  5584.6  433.01  5670.2  436.25
#Mann=5,-1,0
  4516.3   0.035       0  4836.0    0.05       0  4985.6   0.035       0
  4995.3    0.05       0  5082.3    0.05       0
Bank Sta=4985.6,4995.3
Exp/Cntr=0.3,0.1

Type RM Length L Ch R = 1,24927,259,259,259
BEGIN DESCRIPTION:
Mill Creek24927.43
END DESCRIPTION:
XS GIS Cut Line= 3
      2754025.26      6820056.25      2754203.67      6820337.66
      2754515.66      6820930.59
#Sta/Elev= 30
  4669.3  440.14  4711.6  438.02  4738.0  436.00  4789.7  433.53  4810.9  431.48
  4862.6  428.27  4889.7  425.61  4911.7  424.48  4941.4  423.40  4977.8  424.55
  5015.1  424.02  5020.7  418.57  5024.0  416.38  5024.5  415.88  5033.2  415.88
  5033.7  416.38  5037.1  418.01  5042.8  425.10  5086.8  423.01  5103.2  423.59
  5235.5  423.65  5340.0  423.08  5384.1  423.81  5400.5  424.37  5406.1  425.76
  5413.1  425.13  5458.3  429.51  5516.3  433.72  5582.6  434.07  5672.5  437.96
#Mann=4,-1,0
  4669.3   0.035       0  4711.6    0.16       0  5024.0    0.07       0
  5033.7    0.05       0
Bank Sta=5024,5033.7
Exp/Cntr=0.3,0.1

Type RM Length L Ch R = 1,24668,245,245,245
BEGIN DESCRIPTION:
Mill Creek24668.09
END DESCRIPTION:
XS GIS Cut Line= 3
      2753964.40      6820141.38      2753984.05      6820422.40
      2754001.12      6821174.40
#Sta/Elev= 30
  4729.9  440.34  4769.6  437.81  4822.9  433.20  4829.8  432.26  4844.7  431.23
  4889.9  427.82  4899.9  427.41  4910.0  426.16  4943.0  423.84  4966.5  422.32
  5000.2  423.15  5011.6  422.31  5015.4  416.67  5015.9  416.17  5024.6  416.17
  5025.1  416.67  5032.1  419.23  5040.2  423.03  5050.2  423.50  5060.2  422.96
  5130.2  421.46  5150.2  420.68  5180.3  420.78  5190.3  421.54  5220.3  420.91
  5260.3  421.16  5390.3  423.48  5670.4  427.21  5740.4  430.03  5763.8  431.87
#Mann=7,-1,0
  4729.9   0.035       0  4822.9    0.16       0  4844.7   0.035       0
  4943.0    0.16       0  5015.4    0.07       0  5025.1    0.16       0
  5032.1    0.05       0
Bank Sta=5015.4,5025.1
Exp/Cntr=0.3,0.1

Type RM Length L Ch R = 1,24423,241,241,241
BEGIN DESCRIPTION:
Mill Creek24423.38
END DESCRIPTION:
XS GIS Cut Line= 3
      2753764.26      6820150.40      2753770.15      6820514.20
      2753784.67      6821247.40
#Sta/Elev= 30
  4641.6  436.90  4742.2  430.27  4772.2  428.82  4782.2  427.72  4867.5  421.98
  4892.2  420.51  4913.9  420.87  4962.2  421.47  4972.2  419.76  4977.3  413.89
  4977.8  413.39  4986.6  413.39  4987.1  413.89  4992.3  419.92  5001.4  421.85
  5047.9  420.84  5087.4  420.86  5152.3  420.02  5162.3  420.62  5202.3  419.81
  5212.3  420.20  5262.3  419.46  5312.3  419.54  5402.3  421.62  5422.3  423.19
  5492.3  426.40  5562.4  430.82  5662.4  434.74  5722.4  438.23  5738.8  439.77
#Mann=7,-1,0
  4641.6   0.035       0  4742.2    0.16       0  4867.5    0.12       0
  4913.9    0.16       0  4977.3    0.07       0  4987.1    0.16       0
  5087.4    0.05       0
Bank Sta=4977.3,4987.1
Exp/Cntr=0.3,0.1

Type RM Length L Ch R = 1,24182,277,277,277
BEGIN DESCRIPTION:
Mill Creek24181.7
END DESCRIPTION:
XS GIS Cut Line= 3
      2753521.58      6820078.18      2753528.65      6820514.82
      2753530.61      6821041.32
#Sta/Elev= 30
  4567.5  431.96  4620.3  429.90  4660.3  427.05  4734.6  423.33  4770.3  421.65
  4780.3  420.53  4822.5  419.10  4840.4  418.22  4958.9  420.06  5004.2  421.17
  5010.4  417.99  5015.5  412.89  5016.0  412.39  5024.8  412.39  5025.3  412.89
  5030.4  421.03  5040.1  420.95  5100.4  419.31  5190.4  419.00  5240.4  417.45
  5260.4  418.48  5280.4  417.96  5300.4  418.28  5320.4  419.13  5340.4  420.60
  5360.4  422.99  5450.4  428.76  5470.4  429.63  5500.4  429.69  5530.7  430.55
#Mann=7,-1,0
  4567.5   0.035       0  4734.6    0.16       0  4822.5    0.12       0
  4958.9    0.16       0  5015.5    0.07       0  5025.3    0.16       0
  5040.1    0.05       0
Bank Sta=5015.5,5025.3
Exp/Cntr=0.3,0.1

Type RM Length L Ch R = 1,23905,277,277,277
BEGIN DESCRIPTION:
Mill Creek23905.33
END DESCRIPTION:
XS GIS Cut Line= 3
      2753234.02      6819811.47      2753268.66      6820567.41
      2753274.88      6821157.94
#Sta/Elev= 30
  4249.8  429.27  4349.4  427.00  4379.5  425.42  4403.4  425.35  4449.5  423.63
  4499.6  423.01  4599.7  418.71  4677.6  417.22  4719.8  416.82  4779.9  417.77
  4856.2  417.68  4917.9  418.00  4980.1  419.66  4995.2  413.35  4995.7  412.85
  5004.5  412.85  5005.0  413.35  5005.8  419.38  5080.1  418.68  5100.1  417.91
  5120.1  415.63  5130.1  415.82  5140.1  417.14  5167.9  417.56  5210.1  420.78
  5232.0  420.88  5270.1  422.89  5340.1  424.39  5500.2  425.46  5597.1  427.28
#Mann=7,-1,0
  4249.8   0.035       0  4677.6    0.16       0  4856.2    0.12       0
  4917.9    0.16       0  4995.2    0.07       0  5005.0    0.16       0
  5167.9    0.05       0
Bank Sta=4995.2,5005
Exp/Cntr=0.3,0.1

Type RM Length L Ch R = 1,23628,274,274,274
BEGIN DESCRIPTION:
Mill Creek23628.119
END DESCRIPTION:
XS GIS Cut Line= 3
      2753003.31      6819625.78      2753076.31      6820711.33
      2753100.45      6821200.63
#Sta/Elev= 30
  3912.0  426.56  4024.6  422.65  4166.3  419.93  4251.4  418.49  4358.2  416.79
  4509.2  416.49  4718.0  417.05  4795.2  417.19  4816.3  417.07  4869.4  417.19
  4929.5  418.17  4949.6  417.83  4969.6  418.37  4979.6  417.18  4992.3  412.42
  4992.8  411.92  5001.8  411.92  5002.3  412.42  5019.7  417.74  5049.7  417.45
  5062.6  416.71  5089.8  416.35  5119.8  418.24  5179.9  417.83  5199.9  418.28
  5290.0  420.95  5301.5  422.20  5320.1  421.67  5370.1  422.62  5489.9  426.92
#Mann=10,-1,0
  3912.0    0.05       0  4166.3   0.035       0  4251.4    0.07       0
  4509.2    0.16       0  4718.0    0.12       0  4795.2    0.16       0
  4816.3    0.12       0  4992.3    0.07       0  5002.3    0.12       0
  5062.6    0.05       0
Bank Sta=4992.3,5002.3
Exp/Cntr=0.3,0.1

Type RM Length L Ch R = 1,23354,273,273,273
BEGIN DESCRIPTION:
Mill Creek23353.62
END DESCRIPTION:
XS GIS Cut Line= 3
      2752716.37      6819940.96      2752836.40      6820813.26
      2752914.93      6821213.51
#Sta/Elev= 30
  4121.4  433.13  4183.7  430.15  4228.1  427.75  4233.1  428.26  4252.7  427.43
  4300.1  424.34  4305.1  424.74  4368.8  420.55  4377.1  420.83  4464.6  416.01
  4509.3  415.96  4513.8  415.94  4670.2  414.17  4686.7  413.37  4696.8  414.19
  4757.4  414.79  4806.8  414.37  4828.0  415.45  4858.3  415.00  4969.4  416.10
  4979.4  415.60  4984.5  410.82  4985.0  410.32  4994.6  410.82  4998.3  411.90
  5001.9  411.90  5009.8  415.66  5103.1  415.43  5274.8  420.60  5409.8  425.90
#Mann=9,-1,0
  4121.4    0.05       0  4183.7    0.07       0  4368.8    0.16       0
  4509.3    0.05       0  4513.8    0.16       0  4806.8    0.12       0
  4984.5    0.07       0  4994.6    0.12       0  5103.1    0.05       0
Bank Sta=4984.5,4994.6
Exp/Cntr=0.3,0.1

Type RM Length L Ch R = 1,23081,320,320,320
BEGIN DESCRIPTION:
Mill Creek23081.367
END DESCRIPTION:
XS GIS Cut Line= 3
      2752445.11      6819851.33      2752582.03      6820876.38
      2752626.64      6821220.35
#Sta/Elev= 30
  3981.2  434.12  4088.1  427.92  4112.0  426.41  4255.3  419.91  4334.0  417.32
  4364.2  416.86  4424.8  414.44  4453.0  414.11  4474.5  413.79  4479.5  412.95
  4525.7  413.82  4545.8  413.32  4625.7  413.78  4651.2  413.24  4687.1  412.85
  4750.3  413.55  4860.1  413.38  4909.0  413.85  4928.1  413.40  4989.7  414.93
  4994.8  410.17  4995.3  409.67  5004.4  409.67  5004.9  410.17  5006.2  414.05
  5011.3  415.13  5030.1  413.98  5060.3  413.74  5164.5  415.25  5362.2  424.31
#Mann=7,-1,0
  3981.2    0.05       0  4088.1    0.07       0  4453.0    0.05       0
  4651.2    0.16       0  4750.3    0.05       0  4994.8    0.05       0
  5004.9    0.05       0
Bank Sta=4994.8,5004.9
Exp/Cntr=0.3,0.1

Type RM Length L Ch R = 1,22761,285,285,285
BEGIN DESCRIPTION:
Mill Creek22761.135
END DESCRIPTION:
XS GIS Cut Line= 3
      2752137.04      6820311.46      2752276.00      6820811.00
      2752351.01      6821086.05
#Sta/Elev= 30
  4481.6  425.66  4522.6  424.10  4543.4  422.34  4564.2  421.83  4584.9  419.70
  4649.0  416.12  4709.5  414.08  4762.1  411.33  4796.3  411.98  4813.3  410.64
  4835.7  412.26  4904.2  410.66  4917.1  412.30  4943.6  412.64  4983.0  414.37
  4989.7  410.42  4992.5  407.89  4993.0  407.39  5002.1  407.39  5002.6  407.89
  5010.5  412.30  5017.4  413.71  5051.9  412.72  5072.7  413.61  5114.1  417.14
  5166.0  419.98  5197.0  422.55  5210.9  425.03  5269.6  427.48  5285.2  427.61
#Mann=3,-1,0
  4481.6    0.05       0  4992.5    0.05       0  5002.6    0.05       0
Bank Sta=4992.5,5002.6
Exp/Cntr=0.3,0.1

Type RM Length L Ch R = 1,22476,108,108,108
BEGIN DESCRIPTION:
Mapping XS 94bac7dd
END DESCRIPTION:
XS GIS Cut Line= 4
      2752025.69      6820367.25      2752007.10      6820862.93
      2752010.63      6820899.38      2752311.76      6821090.65
#Sta/Elev= 30
  4505.9  429.39  4539.7  427.65  4549.7  426.39  4569.7  425.62  4619.7  422.05
  4632.8  422.04  4639.7  421.24  4739.8  415.83  4849.9  411.70  4901.3  411.43
  4919.9  410.56  4930.0  409.45  4940.0  410.30  4970.0  408.28  4974.8  406.25
  4975.3  405.75  4984.7  405.75  4985.2  406.25  4990.0  412.18  4998.5  412.91
  5010.0  412.21  5020.1  410.63  5036.9  410.69  5044.9  411.56  5056.8  411.86
  5100.3  411.81  5175.2  411.73  5269.4  417.94  5341.1  424.89  5395.3  426.97
#Mann=4,-1,0
  4505.9   0.035       0  4974.8   0.035       0  4985.2   0.035       0
  5100.3    0.05       0
Bank Sta=4974.8,4985.2
Exp/Cntr=0.3,0.1

Type RM Length L Ch R = 1,22368,283,283,283
BEGIN DESCRIPTION:
Mapping XS b4d33517
END DESCRIPTION:
XS GIS Cut Line= 5
      2751925.14      6820421.93      2751898.99      6820865.51
      2751886.46      6820927.55      2751560.04      6821296.34
      2751340.15      6821578.29
#Sta/Elev= 30
  4560.5  428.64  4579.6  427.30  4589.6  427.46  4609.7  425.78  4639.7  425.55
  4669.8  423.47  4689.8  422.94  4729.9  419.98  4739.9  419.92  4769.9  416.83
  4797.9  415.56  4890.1  413.69  4920.2  412.34  4960.3  412.22  4973.0  411.41
  4980.3  409.05  4983.3  405.71  4983.8  405.21  4997.3  405.71  5004.8  405.75
  5010.4  408.79  5020.6  411.66  5045.7  412.91  5092.1  412.14  5184.1  412.47
  5233.5  411.37  5559.7  411.89  5644.7  410.51  5858.2  421.28  5918.2  423.15
#Mann=3,-1,0
  4560.5    0.05       0  4983.3    0.05       0  4997.3    0.05       0
Bank Sta=4983.3,4997.3
Exp/Cntr=0.3,0.1

Type RM Length L Ch R = 1,22085,437,437,437
BEGIN DESCRIPTION:
Mill Creek22084.891
END DESCRIPTION:
XS GIS Cut Line= 3
      2751778.46      6820514.47      2751653.25      6820960.94
      2751226.00      6821710.99
#Sta/Elev= 30
  4536.3  432.67  4561.3  431.43  4566.5  432.57  4600.6  429.06  4605.8  430.33
  4626.2  428.23  4674.0  427.51  4679.2  428.47  4708.1  426.34  4713.3  428.47
  4719.6  427.05  4747.4  425.68  4752.5  426.56  4899.3  421.59  4948.1  415.84
  4958.5  411.60  4972.7  410.60  4989.7  407.08  4990.4  404.32  4990.9  403.82
  5004.5  404.32  5011.6  404.44  5021.0  409.59  5026.8  409.06  5042.6  412.05
  5114.0  411.36  5165.0  410.56  5356.8  411.66  5414.4  410.03  5863.2  430.63
#Mann=5,-1,0
  4536.3    0.05       0  4990.4    0.05       0  5004.5    0.05       0
  5114.0    0.16       0  5165.0    0.05       0
Bank Sta=4990.4,5004.5
Exp/Cntr=0.3,0.1

Type RM Length L Ch R = 1,21648,415,415,415
BEGIN DESCRIPTION:
Mapping XS d8526861
END DESCRIPTION:
XS GIS Cut Line= 3
      2751304.59      6820510.15      2751263.18      6821007.93
      2751174.18      6821649.99
#Sta/Elev= 30
  4510.2  434.23  4711.7  433.67  4795.9  431.47  4802.1  429.91  4808.8  429.39
  4822.1  427.79  4832.2  425.67  4882.3  422.20  4892.4  420.86  4942.5  412.29
  4952.6  410.86  4962.6  410.58  4982.7  406.73  4985.7  403.92  4986.2  403.42
  4999.3  403.42  4999.8  403.92  5002.8  405.04  5008.7  410.45  5023.0  411.28
  5154.1  409.81  5214.7  410.89  5247.1  410.53  5265.2  409.42  5305.6  410.73
  5366.2  411.34  5390.6  412.36  5457.0  416.92  5547.9  424.33  5657.9  428.54
#Mann=5,-1,0
  4510.2    0.05       0  4808.8    0.16       0  4985.7    0.07       0
  4999.8    0.16       0  5023.0    0.05       0
Bank Sta=4985.7,4999.8
Exp/Cntr=0.3,0.1

Type RM Length L Ch R = 1,21233,475,475,475
BEGIN DESCRIPTION:
Mill Creek21233.14
END DESCRIPTION:
XS GIS Cut Line= 3
      2750939.54      6820373.03      2750906.22      6821023.36
      2750878.26      6821694.60
#Sta/Elev= 30
  4361.3  426.36  4459.4  426.79  4526.4  425.77  4531.4  425.09  4619.6  422.27
  4689.7  417.50  4719.2  415.25  4729.7  413.89  4749.8  413.16  4879.9  409.72
  4950.0  410.66  4970.1  406.67  4980.1  403.79  4983.0  402.45  4983.5  401.95
  4996.6  401.95  4997.1  402.45  5008.8  408.05  5012.5  408.05  5020.1  410.28
  5060.2  409.06  5090.2  409.25  5200.3  408.22  5340.4  410.31  5376.8  412.12
  5381.8  411.92  5420.5  415.03  5510.6  420.01  5617.1  424.21  5684.3  426.05
#Mann=3,-1,0
  4361.3    0.05       0  4983.0    0.05       0  4997.1    0.05       0
Bank Sta=4983,4997.1
Exp/Cntr=0.3,0.1

Type RM Length L Ch R = 1,20758,661,661,661
BEGIN DESCRIPTION:
Mill Creek20758.29
END DESCRIPTION:
XS GIS Cut Line= 3
      2750457.82      6820354.42      2750486.44      6820874.69
      2750495.79      6821706.08
#Sta/Elev= 30
  4491.7  427.86  4518.3  428.47  4546.5  428.43  4551.5  427.99  4598.4  429.11
  4638.5  429.21  4658.5  428.61  4688.6  426.76  4778.7  419.81  4858.8  411.99
  4939.0  408.00  4969.0  407.62  4999.0  409.18  5012.0  400.76  5012.5  400.26
  5025.7  400.26  5026.2  400.76  5029.1  408.70  5069.1  409.02  5169.1  407.79
  5239.1  407.69  5259.1  406.99  5359.1  412.24  5399.1  413.46  5459.1  416.75
  5499.1  417.78  5539.1  419.85  5659.1  423.65  5729.1  424.55  5844.2  427.64
#Mann=3,-1,0
  4491.7    0.05       0  5012.0    0.05       0  5026.2    0.05       0
Bank Sta=5012,5026.2
Exp/Cntr=0.3,0.1

Type RM Length L Ch R = 1,20097,440,440,440
BEGIN DESCRIPTION:
Mill Creek20097.08
END DESCRIPTION:
XS GIS Cut Line= 3
      2750047.32      6820552.40      2750044.06      6821175.76
      2750087.31      6821821.04
#Sta/Elev= 30
  4390.7  426.83  4426.3  426.68  4459.3  425.65  4539.3  425.28  4609.3  426.17
  4659.3  424.72  4679.3  423.74  4699.3  421.56  4819.3  411.96  4909.3  406.59
  4989.3  407.50  4999.3  406.03  5001.9  399.75  5002.4  399.25  5016.0  399.25
  5016.5  399.75  5019.3  399.83  5029.3  405.88  5039.4  406.79  5049.4  405.93
  5059.4  406.45  5089.5  406.28  5099.5  406.87  5169.7  406.93  5259.9  411.27
  5266.1  412.19  5360.1  418.35  5430.2  422.06  5630.7  426.66  5660.8  426.14
#Mann=4,-1,0
  4390.7    0.16       0  4426.3    0.05       0  5001.9    0.05       0
  5016.5    0.05       0
Bank Sta=5001.9,5016.5
Exp/Cntr=0.3,0.1

Type RM Length L Ch R = 1,19657,615,615,615
BEGIN DESCRIPTION:
Mill Creek19657.45
END DESCRIPTION:
XS GIS Cut Line= 3
      2749983.28      6820480.26      2749638.96      6821043.47
      2749310.70      6821502.69
#Sta/Elev= 30
  4353.7  428.07  4438.6  424.87  4520.5  417.42  4577.3  412.53  4753.1  405.18
  4765.7  403.84  4808.5  405.07  4928.1  407.15  4940.6  405.69  4949.4  404.05
  4964.0  404.88  4970.7  407.07  4999.2  405.03  5000.1  397.86  5000.6  397.36
  5014.8  397.86  5022.2  399.42  5028.4  403.40  5035.4  399.85  5043.1  400.75
  5049.3  404.51  5057.9  403.27  5064.0  405.56  5141.7  406.91  5221.3  410.88
  5280.3  412.21  5286.4  413.54  5330.4  415.20  5465.6  425.26  5578.3  424.60
#Mann=7,-1,0
  4353.7    0.16       0  4520.5    0.05       0  4808.5    0.12       0
  4940.6    0.16       0  5000.1    0.07       0  5014.8    0.16       0
  5141.7    0.05       0
Bank Sta=5000.1,5014.8
Exp/Cntr=0.3,0.1

Type RM Length L Ch R = 1,19042,438,438,438
BEGIN DESCRIPTION:
Mill Creek19042.25
END DESCRIPTION:
XS GIS Cut Line= 3
      2749855.02      6820129.10      2749496.45      6820551.67
      2749129.81      6820993.32
#Sta/Elev= 30
  4460.6  426.15  4553.9  426.98  4673.6  425.96  4745.0  421.93  4759.3  420.01
  4765.9  420.54  4779.4  419.65  4847.0  412.83  4894.5  407.78  4915.3  403.44
  4979.0  403.02  4985.9  395.33  4986.4  394.83  5000.6  395.33  5007.6  396.27
  5011.3  403.23  5021.9  404.02  5042.7  403.04  5064.9  404.71  5092.2  403.17
  5114.3  404.65  5143.0  405.05  5178.1  408.58  5213.3  409.99  5241.9  413.95
  5284.7  415.80  5433.4  425.27  5497.2  428.37  5519.3  427.62  5588.8  428.24
#Mann=6,-1,0
  4460.6    0.16       0  4779.4    0.12       0  4847.0    0.16       0
  4985.9    0.07       0  5000.6    0.16       0  5284.7    0.05       0
Bank Sta=4985.9,5000.6
Exp/Cntr=0.3,0.1

Type RM Length L Ch R = 1,18604,432,432,432
BEGIN DESCRIPTION:
Mill Creek18603.54
END DESCRIPTION:
XS GIS Cut Line= 3
      2749570.02      6819878.02      2749233.47      6820301.15
      2748914.18      6820740.30
#Sta/Elev= 30
  4482.0  427.34  4608.1  424.84  4672.1  420.51  4708.1  416.07  4728.1  413.72
  4785.9  408.69  4864.4  405.53  4901.8  402.88  4942.8  403.74  4963.7  402.80
  4978.1  397.63  4984.5  395.04  4985.2  394.12  4985.7  393.62  4999.9  394.12
  5006.9  402.40  5013.3  404.12  5063.3  403.14  5103.3  404.09  5149.1  406.51
  5214.0  412.41  5299.8  418.57  5306.8  417.15  5314.5  419.04  5320.7  418.02
  5370.9  420.92  5379.4  422.24  5385.6  421.88  5400.3  423.71  5565.6  425.30
#Mann=7,-1,0
  4482.0    0.12       0  4708.1    0.16       0  4728.1    0.12       0
  4901.8    0.16       0  4985.2    0.07       0  4999.9    0.16       0
  5103.3    0.05       0
Bank Sta=4985.2,4999.9
Exp/Cntr=0.3,0.1

Type RM Length L Ch R = 1,18172,365,365,365
BEGIN DESCRIPTION:
Mill Creek18171.67
END DESCRIPTION:
XS GIS Cut Line= 3
      2749150.34      6819540.62      2748955.51      6820123.01
      2748776.16      6820612.26
#Sta/Elev= 30
  4397.5  424.65  4525.6  422.78  4551.9  420.02  4615.1  416.74  4620.3  417.38
  4646.6  414.62  4651.9  415.60  4688.5  412.22  4741.4  406.98  4804.5  402.95
  4873.0  401.12  4925.1  402.39  4956.8  400.06  4967.7  402.09  4986.8  401.51
  4994.0  400.57  4999.3  401.39  5007.9  393.91  5017.7  393.38  5018.2  392.88
  5032.5  393.38  5041.4  400.63  5062.7  406.61  5116.6  410.97  5147.9  415.27
  5212.4  419.01  5289.0  421.64  5356.8  422.36  5407.2  422.76  5532.7  423.30
#Mann=8,-1,0
  4397.5    0.16       0  4688.5    0.12       0  4986.8    0.16       0
  5017.7    0.07       0  5032.5    0.16       0  5212.4    0.05       0
  5356.8    0.16       0  5407.2    0.05       0
Bank Sta=5017.7,5032.5
Exp/Cntr=0.3,0.1

Type RM Length L Ch R = 1,17807,282,282,282
BEGIN DESCRIPTION:
Mill Creek17806.98
END DESCRIPTION:
XS GIS Cut Line= 3
      2748832.58      6819366.74      2748687.11      6819913.93
      2748546.19      6820456.01
#Sta/Elev= 30
  4437.5  420.62  4485.5  418.57  4521.3  415.51  4566.1  413.16  4595.6  413.27
  4600.8  411.99  4669.6  408.55  4676.0  409.76  4681.1  408.34  4710.9  410.27
  4833.8  410.99  4911.7  408.56  4959.3  400.87  4969.6  400.29  4979.4  393.51
  4979.9  393.01  4994.3  393.51  5003.7  393.59  5011.0  400.02  5021.3  400.93
  5042.0  398.07  5052.3  399.50  5067.8  398.58  5073.0  401.22  5151.8  403.38
  5279.6  409.44  5305.8  412.46  5321.0  411.55  5503.4  422.73  5563.8  423.76
#Mann=6,-1,0
  4437.5    0.12       0  4521.3    0.16       0  4833.8    0.12       0
  4979.4    0.07       0  4994.3    0.12       0  5151.8    0.05       0
Bank Sta=4979.4,4994.3
Exp/Cntr=0.3,0.1

Type RM Length L Ch R = 1,17525,266,266,266
BEGIN DESCRIPTION:
Mill Creek17525.23
END DESCRIPTION:
XS GIS Cut Line= 3
      2748551.37      6819323.59      2748419.00      6819876.31
      2748310.98      6820335.84
#Sta/Elev= 30
  4443.9  422.75  4508.1  423.01  4605.8  422.31  4677.7  414.96  4718.9  409.67
  4740.3  408.28  4780.6  406.26  4787.3  405.00  4829.4  401.93  4883.4  399.61
  4924.5  400.97  4955.4  400.37  4960.6  399.28  4965.8  391.79  4978.8  390.69
  4979.3  390.19  4993.7  390.69  5002.7  391.63  5007.8  397.59  5009.8  398.40
  5012.1  399.33  5034.9  400.24  5087.4  400.99  5138.2  407.07  5191.7  413.11
  5267.2  418.12  5335.5  420.09  5366.3  422.41  5399.6  421.66  5484.3  423.93
#Mann=8,-1,0
  4443.9    0.12       0  4508.1    0.16       0  4740.3    0.12       0
  4978.8    0.07       0  4993.7    0.12       0  5009.8    0.16       0
  5034.9    0.12       0  5138.2    0.05       0
Bank Sta=4978.8,4993.7
Exp/Cntr=0.3,0.1

Type RM Length L Ch R = 1,17259,720,720,720
BEGIN DESCRIPTION:
Mill Creek17258.59
END DESCRIPTION:
XS GIS Cut Line= 3
      2748337.09      6819063.89      2748211.05      6819720.65
      2748080.96      6820179.83
#Sta/Elev= 30
  4339.7  421.34  4414.1  415.91  4509.9  409.74  4520.0  405.89  4528.2  406.48
  4533.3  405.12  4540.2  406.22  4550.6  408.92  4637.2  410.57  4683.0  409.50
  4764.4  403.13  4818.8  400.68  4852.7  399.49  4886.6  399.74  4902.2  397.83
  4927.3  399.83  4968.1  399.96  4988.4  398.71  4998.6  396.23  5003.9  390.35
  5004.4  389.85  5018.8  390.35  5029.6  398.27  5045.3  400.13  5112.7  403.01
  5183.8  410.77  5191.4  412.73  5216.7  414.81  5337.5  420.32  5485.7  419.96
#Mann=8,-1,0
  4339.7    0.16       0  4414.1    0.12       0  4540.2    0.16       0
  4818.8    0.12       0  4852.7    0.16       0  5003.9    0.07       0
  5018.8    0.16       0  5183.8    0.05       0
Bank Sta=5003.9,5018.8
Exp/Cntr=0.3,0.1

Type RM Length L Ch R = 1,16539,651,651,651
BEGIN DESCRIPTION:
Mill Creek16539.142
END DESCRIPTION:
XS GIS Cut Line= 3
      2748200.96      6819036.03      2747956.56      6819190.45
      2747382.11      6819912.91
#Sta/Elev= 30
  4710.9  422.07  4797.6  421.04  4856.7  416.27  4941.5  407.34  4965.2  406.11
  4972.0  404.06  4977.9  396.59  4985.8  388.94  4986.3  388.44  5000.7  388.94
  5003.5  389.50  5008.0  395.30  5022.4  397.15  5028.8  396.23  5036.9  398.14
  5078.5  396.54  5179.4  399.01  5235.5  399.53  5297.1  398.02  5307.3  399.06
  5343.3  398.86  5378.0  399.91  5435.1  399.37  5605.5  407.17  5704.8  407.73
  5748.1  410.16  5805.6  410.55  5826.6  412.64  5841.0  411.82  5923.0  414.03
#Mann=7,-1,0
  4710.9    0.16       0  4797.6    0.12       0  4985.8    0.07       0
  5000.7    0.12       0  5179.4    0.05       0  5297.1    0.16       0
  5343.3    0.05       0
Bank Sta=4985.8,5000.7
Exp/Cntr=0.3,0.1

Type RM Length L Ch R = 1,15888,324,324,324
BEGIN DESCRIPTION:
Mill Creek15887.788
END DESCRIPTION:
XS GIS Cut Line= 3
      2747501.00      6818135.96      2747451.01      6819161.55
      2747336.43      6819892.62
#Sta/Elev= 30
  3973.2  434.94  4031.0  433.49  4208.5  422.83  4383.9  402.48  4423.0  399.80
  4591.7  398.16  4599.0  391.19  4609.0  391.62  4619.0  398.53  4658.0  397.79
  4801.3  397.38  4824.8  397.54  4977.5  396.13  4989.4  395.74  4997.2  389.05
  5002.0  387.54  5002.5  387.04  5017.1  387.54  5019.7  393.69  5039.9  397.17
  5110.8  400.86  5157.2  401.34  5283.0  402.60  5424.6  405.04  5444.8  406.55
  5518.7  406.43  5576.3  409.75  5616.9  409.62  5657.4  412.66  5740.0  414.32
#Mann=11,-1,0
  3973.2    0.07       0  4031.0    0.16       0  4423.0    0.12       0
  4658.0    0.16       0  4801.3    0.12       0  4824.8    0.16       0
  4977.5    0.12       0  5002.0    0.07       0  5017.1    0.12       0
  5157.2    0.16       0  5283.0    0.05       0
Bank Sta=5002,5017.1
Exp/Cntr=0.3,0.1

Type RM Length L Ch R = 1,15564,285,285,285
BEGIN DESCRIPTION:
Mill Creek15563.993
END DESCRIPTION:
XS GIS Cut Line= 3
      2747321.90      6818110.26      2747175.93      6819161.18
      2747059.25      6819865.17
#Sta/Elev= 30
  3939.0  425.31  4060.9  425.09  4135.0  421.34  4290.5  402.49  4394.1  396.54
  4464.7  397.18  4474.8  388.97  4484.9  388.12  4495.0  393.59  4505.1  395.42
  4528.7  396.62  4575.8  394.30  4595.3  397.64  4700.3  395.41  4743.7  394.22
  4806.5  395.89  4939.2  397.60  4953.6  395.68  4958.8  394.26  4963.8  396.34
  4972.0  387.41  4972.5  386.91  4987.2  387.41  4997.4  394.45  5010.0  395.57
  5070.8  395.65  5111.3  399.08  5293.4  400.33  5398.7  402.50  5713.6  415.57
#Mann=9,-1,0
  3939.0    0.07       0  4135.0    0.16       0  4290.5    0.12       0
  4700.3    0.16       0  4806.5    0.12       0  4953.6    0.16       0
  4972.0    0.07       0  4987.2    0.16       0  5293.4    0.05       0
Bank Sta=4972,4987.2
Exp/Cntr=0.3,0.1

Type RM Length L Ch R = 1,15279,632,632,632
BEGIN DESCRIPTION:
Mill Creek15278.643
END DESCRIPTION:
XS GIS Cut Line= 3
      2747245.46      6818170.80      2746923.67      6819105.25
      2746670.49      6819729.89
#Sta/Elev= 30
  4011.7  420.54  4115.0  417.13  4178.1  412.86  4195.3  411.39  4245.1  406.56
  4286.9  398.22  4382.1  395.30  4390.7  386.70  4395.9  387.90  4403.2  393.69
  4453.1  396.31  4796.5  393.44  4916.1  396.66  4935.4  390.61  4942.1  390.99
  4947.3  386.44  4973.3  390.33  4978.6  386.77  4984.9  392.83  4995.1  395.43
  5012.7  394.96  5017.0  394.21  5025.9  385.96  5026.4  385.46  5041.1  385.96
  5070.9  394.86  5111.2  398.64  5377.7  403.91  5556.5  408.48  5674.0  414.94
#Mann=8,-1,0
  4011.7    0.07       0  4178.1    0.16       0  4195.3    0.12       0
  4935.4    0.16       0  5012.7    0.12       0  5025.9    0.07       0
  5041.1    0.12       0  5377.7    0.05       0
Bank Sta=5025.9,5041.1
Exp/Cntr=0.3,0.1

Type RM Length L Ch R = 1,14647,268,268,268
BEGIN DESCRIPTION:
Mill Creek14647.169
END DESCRIPTION:
XS GIS Cut Line= 3
      2747175.99      6818261.01      2746753.53      6818738.57
      2746300.99      6819436.02
#Sta/Elev= 30
  4362.4  413.34  4454.8  406.45  4553.5  395.32  4589.4  396.47  4755.2  395.34
  4886.4  395.34  4914.9  392.69  4936.5  395.56  4971.8  394.47  4977.2  385.25
  4977.7  384.75  4994.7  385.25  5002.3  385.30  5021.9  394.14  5058.2  395.13
  5079.3  394.02  5086.3  392.78  5094.4  394.02  5100.4  393.16  5130.7  395.29
  5194.0  393.77  5224.3  396.14  5315.2  398.46  5447.7  399.72  5520.3  401.67
  5527.4  402.61  5586.8  401.97  5622.8  403.42  5665.3  403.23  5831.4  409.14
#Mann=6,-1,0
  4362.4    0.07       0  4454.8    0.12       0  4755.2    0.16       0
  4977.2    0.07       0  4994.7    0.16       0  5315.2    0.05       0
Bank Sta=4977.2,4994.7
Exp/Cntr=0.3,0.1

Type RM Length L Ch R = 1,14379,883,883,883
BEGIN DESCRIPTION:
Mill Creek14379.07
END DESCRIPTION:
XS GIS Cut Line= 3
      2747150.92      6818251.64      2746619.52      6818524.64
      2745866.66      6819389.82
#Sta/Elev= 30
  4410.1  409.92  4492.2  404.78  4570.1  395.20  4643.2  394.50  4732.9  394.14
  4898.3  394.28  4955.3  394.60  4969.4  392.44  4986.0  392.47  4991.6  391.29
  4997.9  383.57  4998.4  383.07  5015.4  383.57  5035.8  385.42  5064.3  385.29
  5070.9  390.20  5078.5  393.34  5135.3  392.73  5170.6  394.47  5199.1  393.46
  5248.4  394.75  5354.8  397.98  5440.1  395.92  5652.2  399.21  5709.0  402.46
  5907.4  403.96  5957.1  406.79  5999.5  406.87  6070.7  411.31  6154.4  414.54
#Mann=8,-1,0
  4410.1    0.07       0  4492.2    0.12       0  4643.2    0.16       0
  4732.9    0.12       0  4898.3    0.16       0  4997.9    0.07       0
  5015.4    0.16       0  5248.4    0.05       0
Bank Sta=4997.9,5015.4
Exp/Cntr=0.3,0.1

Type RM Length L Ch R = 1,13496,461,461,461
BEGIN DESCRIPTION:
Mill Creek13496.25
END DESCRIPTION:
XS GIS Cut Line= 3
      2745968.09      6817734.93      2745964.08      6818269.93
      2745936.65      6819230.43
#Sta/Elev= 30
  4474.5  418.59  4531.8  416.79  4630.6  413.93  4738.8  412.74  4770.6  411.16
  4846.6  404.32  4890.6  399.54  4910.6  395.06  4930.6  391.92  4950.6  390.83
  4960.6  385.45  4970.6  383.94  4971.7  382.18  4972.2  381.68  4989.4  382.18
  4990.6  385.38  5007.5  392.66  5042.4  393.49  5238.2  391.69  5441.4  393.61
  5500.8  393.95  5570.8  396.85  5590.8  398.87  5730.9  399.34  5790.9  400.45
  5810.9  401.87  5822.0  401.16  5921.0  404.22  5961.0  406.91  5970.4  406.59
#Mann=9,-1,0
  4474.5    0.16       0  4531.8    0.07       0  4738.8    0.16       0
  4846.6    0.12       0  4971.7    0.07       0  4989.4    0.12       0
  5042.4    0.16       0  5238.2    0.07       0  5441.4    0.05       0
Bank Sta=4971.7,4989.4
Exp/Cntr=0.3,0.1

Type RM Length L Ch R = 1,13035,336,336,336
BEGIN DESCRIPTION:
Mill Creek13035.17
END DESCRIPTION:
XS GIS Cut Line= 3
      2745491.73      6817552.05      2745536.28      6818270.07
      2745699.38      6819193.57
#Sta/Elev= 30
  4289.6  413.58  4348.7  410.88  4408.8  401.60  4436.6  395.53  4441.6  396.71
  4499.0  388.39  4529.0  390.31  4539.0  388.21  4597.5  389.89  4639.2  387.99
  4669.3  390.62  4689.3  388.27  4729.4  390.99  4939.8  392.30  4949.8  391.88
  4959.8  384.66  4961.0  381.05  4961.5  380.55  4978.8  381.05  4989.9  389.24
  5020.1  391.47  5089.9  390.12  5131.8  392.09  5231.8  391.58  5243.5  389.79
  5390.5  393.87  5456.8  397.99  5553.4  401.06  5671.9  400.93  5946.8  410.98
#Mann=5,-1,0
  4289.6    0.12       0  4961.0    0.07       0  4978.8    0.12       0
  5231.8    0.16       0  5390.5    0.05       0
Bank Sta=4961,4978.8
Exp/Cntr=0.3,0.1

Type RM Length L Ch R = 1,12699,286,286,286
BEGIN DESCRIPTION:
Mill Creek12698.658
END DESCRIPTION:
XS GIS Cut Line= 3
      2745389.84      6817544.18      2745245.84      6818131.38
      2744686.40      6818596.76
#Sta/Elev= 30
  4395.4  409.36  4442.7  409.09  4464.2  408.93  4477.1  404.76  4484.8  399.81
  4513.5  389.17  4546.6  387.91  4596.7  390.25  4685.0  388.96  4726.6  390.39
  4917.2  390.29  4968.7  391.57  4976.1  391.42  4981.3  387.71  5003.1  384.46
  5006.8  381.55  5012.2  381.01  5012.7  380.51  5030.0  381.01  5035.4  390.77
  5041.9  391.51  5134.3  388.78  5170.9  389.20  5411.7  390.59  5524.9  393.14
  5546.1  395.44  5574.4  395.44  5610.9  399.20  5646.0  400.33  5727.7  407.27
#Mann=5,-1,0
  4395.4    0.16       0  4442.7    0.12       0  5012.2    0.07       0
  5030.0    0.12       0  5170.9    0.05       0
Bank Sta=5012.2,5030
Exp/Cntr=0.3,0.1

Type RM Length L Ch R = 1,12413,211,211,211
BEGIN DESCRIPTION:
Mill Creek12412.92
END DESCRIPTION:
XS GIS Cut Line= 3
      2745275.98      6817461.04      2745026.00      6817961.00
      2744526.00      6818661.00
#Sta/Elev= 30
  4440.8  412.18  4460.6  411.38  4485.5  410.36  4574.9  401.62  4642.0  393.18
  4717.5  388.54  4723.1  389.55  4731.4  388.12  4776.2  389.05  4829.3  388.04
  4834.9  389.32  4843.2  388.13  4888.0  387.83  4941.1  389.11  4963.4  388.01
  4985.8  391.18  5002.8  391.29  5013.3  382.21  5019.1  380.50  5019.6  380.00
  5037.0  380.50  5048.9  390.99  5114.1  388.88  5208.9  389.39  5407.8  391.16
  5523.3  396.11  5573.7  399.88  5638.8  401.49  5716.2  406.87  5860.0  411.63
#Mann=5,-1,0
  4440.8    0.16       0  4460.6    0.12       0  5019.1    0.07       0
  5037.0    0.12       0  5208.9    0.05       0
Bank Sta=5019.1,5037
Exp/Cntr=0.3,0.1

Type RM Length L Ch R = 1,12202,238,238,238
BEGIN DESCRIPTION:
Mill Creek12201.79
END DESCRIPTION:
XS GIS Cut Line= 3
      2745209.19      6817505.24      2744904.40      6817801.86
      2744396.04      6818402.77
#Sta/Elev= 30
  4583.5  406.98  4745.4  388.83  4787.8  389.49  4816.1  387.38  4837.4  388.70
  4886.8  389.59  4894.0  389.28  4901.0  386.91  4908.1  386.59  4922.3  388.67
  4941.7  389.74  4957.6  386.28  4962.6  380.21  4963.1  379.71  4980.9  380.21
  4985.9  381.68  4992.8  381.31  5000.0  385.50  5011.4  384.85  5014.1  390.38
  5020.8  390.79  5149.0  388.59  5255.9  388.26  5291.0  389.98  5319.6  392.82
  5340.5  391.99  5426.4  392.43  5560.2  395.01  5666.8  399.53  5795.9  406.52
#Mann=6,-1,0
  4583.5    0.12       0  4941.7    0.16       0  4962.6    0.07       0
  4980.9    0.16       0  5149.0    0.07       0  5426.4    0.05       0
Bank Sta=4962.6,4980.9
Exp/Cntr=0.3,0.1

Type RM Length L Ch R = 1,11964,630,630,630
BEGIN DESCRIPTION:
Mill Creek11964.38
END DESCRIPTION:
XS GIS Cut Line= 3
      2745226.00      6817461.00      2744726.00      6817661.00
      2744126.03      6818260.97
#Sta/Elev= 30
  4462.6  410.92  4560.9  401.79  4633.6  393.97  4645.7  391.61  4656.5  387.29
  4663.2  386.67  4678.0  388.72  4741.3  387.99  4776.3  389.01  4807.3  388.30
  4880.9  389.14  4979.6  389.18  4986.3  387.76  4989.3  379.64  4989.8  379.14
  5007.6  379.64  5029.4  388.69  5043.5  389.48  5057.7  389.40  5100.1  386.58
  5128.4  388.52  5142.5  387.09  5170.7  388.39  5199.1  388.13  5227.4  389.59
  5300.2  388.87  5397.1  388.83  5566.8  391.65  5694.1  396.59  5849.6  405.67
#Mann=6,-1,0
  4462.6    0.12       0  4880.9    0.16       0  4989.3    0.07       0
  5007.6    0.16       0  5170.7    0.07       0  5300.2    0.05       0
Bank Sta=4989.3,5007.6
Exp/Cntr=0.3,0.1

Type RM Length L Ch R = 1,11334,768,768,768
BEGIN DESCRIPTION:
Mill Creek11333.748
END DESCRIPTION:
XS GIS Cut Line= 5
      2745195.45      6817323.00      2744575.64      6817494.38
      2744301.00      6817636.00      2744162.12      6817761.56
      2743771.62      6818154.81
#Sta/Elev= 30
  3860.7  411.24  4007.7  398.71  4119.5  390.21  4134.9  386.08  4161.0  388.47
  4233.6  386.82  4316.6  388.46  4337.4  386.23  4361.5  389.43  4378.1  388.61
  4454.9  388.26  4738.3  388.05  4933.1  388.11  4940.5  387.60  4947.3  384.74
  4952.3  378.67  4952.8  378.17  4970.7  378.67  4975.7  387.10  4982.4  387.97
  5003.9  386.38  5011.0  383.44  5039.3  387.56  5046.4  386.55  5137.1  390.23
  5203.4  392.89  5281.7  398.62  5328.0  401.45  5442.3  407.72  5554.2  410.71
#Mann=11,-1,0
  3860.7    0.16       0  4007.7    0.12       0  4378.1    0.16       0
  4454.9    0.05       0  4738.3    0.16       0  4952.3    0.07       0
  4970.7    0.16       0  5137.1    0.05       0  5203.4    0.16       0
  5281.7    0.12       0  5328.0    0.05       0
Bank Sta=4952.3,4970.7
Exp/Cntr=0.3,0.1

Type RM Length L Ch R = 1,10566,320,320,320
BEGIN DESCRIPTION:
Mill Creek10584.12
END DESCRIPTION:
XS GIS Cut Line= 3
      2745092.95      6817307.54      2743876.83      6817542.44
      2743606.72      6817663.02
#Sta/Elev= 30
  3761.4  402.96  3809.6  398.76  3960.5  388.72  3965.6  386.42  3992.5  388.51
  4074.4  386.51  4114.8  388.50  4121.1  386.33  4126.2  386.20  4145.3  388.36
  4224.2  387.64  4238.3  387.40  4695.3  385.47  4850.5  386.66  4965.6  386.59
  4980.5  384.51  4988.7  377.31  4989.2  376.81  5007.1  377.31  5007.6  383.47
  5013.0  383.11  5022.8  386.38  5077.2  387.41  5088.5  389.18  5105.9  388.31
  5111.4  392.12  5157.8  398.40  5181.0  399.91  5274.5  402.44  5295.8  402.70
#Mann=8,-1,0
  3761.4    0.16       0  3809.6    0.12       0  4224.2    0.16       0
  4238.3    0.05       0  4850.5    0.12       0  4988.7    0.07       0
  5007.1    0.12       0  5274.5    0.05       0
Bank Sta=4988.7,5007.1
Exp/Cntr=0.3,0.1

Type RM Length L Ch R = 1,10246,401,401,401
BEGIN DESCRIPTION:
Mapping XS 338a819f
END DESCRIPTION:
XS GIS Cut Line= 3
      2745053.48      6817289.77      2743825.01      6817296.75
      2743334.16      6817352.55
#Sta/Elev= 30
  3772.3  399.27  3785.0  398.17  3939.8  388.19  4029.8  388.43  4089.8  386.11
  4109.8  388.33  4198.5  387.79  4289.8  386.22  4902.0  384.14  4939.8  386.03
  5002.8  386.19  5009.9  385.46  5010.7  376.63  5011.2  376.13  5029.1  376.63
  5030.0  378.37  5040.0  384.58  5050.1  385.68  5191.0  384.51  5271.5  386.97
  5290.0  389.72  5331.9  394.58  5362.1  394.73  5389.8  392.17  5402.4  390.78
  5432.2  391.01  5442.6  395.16  5462.8  398.16  5489.7  399.33  5494.8  399.39
#Mann=9,-1,0
  3772.3    0.16       0  3785.0    0.12       0  4198.5    0.05       0
  4902.0    0.12       0  5010.7    0.07       0  5029.1    0.12       0
  5290.0    0.16       0  5389.8    0.12       0  5489.7    0.05       0
Bank Sta=5010.7,5029.1
Exp/Cntr=0.3,0.1

Type RM Length L Ch R = 1,9845,494,494,494
BEGIN DESCRIPTION:
Mill Creek10160.664
END DESCRIPTION:
XS GIS Cut Line= 3
      2745083.37      6817261.00      2743627.76      6817017.15
      2743223.62      6817269.40
#Sta/Elev= 30
  3524.1  400.67  3574.0  396.79  3724.2  388.06  3906.7  387.55  3937.1  386.06
  3967.9  386.27  3975.3  387.82  3980.4  386.10  3986.6  387.47  4050.7  387.65
  4352.9  384.77  4434.0  385.16  4616.5  383.53  4837.4  384.47  5004.0  384.79
  5012.3  383.97  5016.4  375.63  5016.9  375.13  5034.8  375.63  5039.5  379.89
  5048.9  384.86  5133.8  383.02  5170.4  384.70  5178.9  383.50  5217.3  384.53
  5264.8  386.70  5280.1  386.15  5335.7  387.35  5411.0  388.66  5476.4  397.34
#Mann=10,-1,0
  3524.1    0.16       0  3574.0    0.12       0  3967.9    0.05       0
  3986.6    0.12       0  4050.7    0.05       0  4837.4    0.12       0
  5016.4    0.07       0  5034.8    0.12       0  5217.3    0.16       0
  5335.7    0.05       0
Bank Sta=5016.4,5034.8
Exp/Cntr=0.3,0.1

Type RM Length L Ch R = 1,9351,439,439,439
BEGIN DESCRIPTION:
Mill Creek9350.683
END DESCRIPTION:
XS GIS Cut Line= 3
      2743826.00      6816310.99      2743676.00      6816661.00
      2743126.03      6817260.97
#Sta/Elev= 30
  4619.2  403.56  4705.8  393.43  4797.0  383.56  4833.2  380.57  4909.3  383.79
  4914.8  380.04  4978.2  382.79  4993.8  376.39  5007.1  375.18  5021.3  383.90
  5042.2  384.38  5049.6  380.69  5056.4  382.22  5063.8  375.17  5070.6  380.02
  5082.6  374.71  5083.1  374.21  5101.8  374.71  5120.5  378.25  5127.3  375.44
  5134.7  379.28  5141.5  375.19  5162.8  375.21  5190.8  384.55  5318.6  383.34
  5401.5  382.98  5486.7  384.75  5547.4  384.52  5707.6  386.83  5813.9  399.01
#Mann=10,-1,0
  4619.2    0.05       0  4705.8    0.12       0  4797.0    0.16       0
  4993.8    0.12       0  5082.6    0.07       0  5101.8    0.12       0
  5318.6    0.16       0  5401.5    0.12       0  5486.7    0.16       0
  5547.4    0.05       0
Bank Sta=5082.6,5101.8
Exp/Cntr=0.3,0.1

Type RM Length L Ch R = 1,8912,429,429,429
BEGIN DESCRIPTION:
Mill Creek8911.782
END DESCRIPTION:
XS GIS Cut Line= 3
      2743725.97      6816111.03      2743476.00      6816361.00
      2742676.01      6817560.98
#Sta/Elev= 30
  4635.3  405.28  4762.5  396.20  4884.0  389.39  4991.8  383.31  4996.3  381.95
  5001.7  373.98  5002.2  373.48  5020.9  373.98  5032.4  379.20  5038.4  378.40
  5047.4  381.27  5053.4  379.93  5060.9  382.94  5075.6  383.12  5085.6  383.19
  5097.0  383.72  5140.5  382.05  5246.6  381.86  5362.5  381.85  5385.5  382.12
  5565.7  384.70  5810.6  384.91  5990.8  388.06  5998.4  388.98  6084.0  390.78
  6192.2  395.99  6207.2  397.88  6222.2  397.03  6372.4  404.28  6431.0  406.01
#Mann=9,-1,0
  4635.3    0.05       0  4884.0    0.12       0  5001.7    0.07       0
  5020.9    0.12       0  5075.6    0.16       0  5085.6    0.12       0
  5246.6    0.05       0  5362.5    0.16       0  5385.5    0.05       0
Bank Sta=5001.7,5020.9
Exp/Cntr=0.3,0.1

Type RM Length L Ch R = 1,8483,302,302,302
BEGIN DESCRIPTION:
Mill Creek8483.199
END DESCRIPTION:
XS GIS Cut Line= 3
      2743626.03      6816010.98      2743176.00      6816311.00
      2742476.01      6817310.98
#Sta/Elev= 30
  4459.7  404.31  4509.3  401.63  4567.9  396.85  4755.7  384.50  4820.3  382.10
  4891.9  382.22  4928.5  383.05  4943.1  381.08  4972.0  380.62  4977.4  373.89
  4977.9  373.39  4996.6  373.89  5003.6  374.11  5008.0  375.33  5014.1  379.79
  5028.9  382.10  5037.2  383.18  5052.9  382.67  5171.9  380.59  5216.4  381.19
  5231.2  379.83  5330.1  382.31  5435.8  382.06  5610.9  383.38  5782.2  386.55
  5913.0  391.69  5963.6  395.93  6013.7  398.87  6102.4  401.87  6221.2  405.05
#Mann=8,-1,0
  4459.7    0.05       0  4891.9    0.16       0  4943.1    0.12       0
  4977.4    0.07       0  4996.6    0.12       0  5052.9    0.16       0
  5435.8    0.05       0  6102.4    0.16       0
Bank Sta=4977.4,4996.6
Exp/Cntr=0.3,0.1

Type RM Length L Ch R = 1,8181,296,296,296
BEGIN DESCRIPTION:
Mill Creek8054.615
END DESCRIPTION:
XS GIS Cut Line= 3
      2743380.09      6815382.13      2742973.73      6816154.56
      2742475.99      6817161.01
#Sta/Elev= 30
  4127.2  410.59  4166.8  411.26  4205.0  410.68  4233.0  408.85  4337.5  398.46
  4453.6  391.20  4491.8  389.96  4535.8  387.21  4767.0  380.77  5000.0  382.19
  5009.5  381.59  5018.3  376.85  5022.3  373.74  5022.8  373.24  5041.5  373.74
  5048.8  382.53  5071.2  381.26  5166.5  379.81  5183.4  380.43  5205.8  377.05
  5219.1  380.62  5375.6  380.91  5452.6  381.16  5519.9  382.84  5682.5  388.69
  5733.0  391.62  5761.7  391.82  5906.9  395.76  6002.2  400.30  6122.8  404.35
#Mann=5,-1,0
  4127.2    0.05       0  5022.3    0.05       0  5041.5    0.05       0
  5375.6    0.05       0  5761.7    0.16       0
Bank Sta=5022.3,5041.5
Exp/Cntr=0.3,0.1

Type RM Length L Ch R = 1,7885,265,265,265
BEGIN DESCRIPTION:
Mapping XS 4701aaff
END DESCRIPTION:
XS GIS Cut Line= 4
      2742709.72      6815132.37      2742873.86      6815647.18
      2742726.03      6816211.08      2742492.99      6816975.86
#Sta/Elev= 30
  3876.7  404.94  4073.9  400.14  4148.8  389.11  4175.8  391.42  4347.6  381.80
  4427.3  383.04  4502.9  380.25  4596.7  381.97  4745.2  380.29  4917.2  380.08
  4968.9  381.46  4977.2  378.98  4982.4  380.07  4986.0  375.36  4987.7  373.14
  4988.2  372.64  5007.1  373.14  5010.4  373.39  5016.4  377.43  5021.7  375.74
  5031.3  379.67  5049.3  378.91  5054.5  380.61  5094.0  380.87  5125.4  379.12
  5191.1  382.63  5229.9  381.27  5294.8  384.56  5562.7  390.43  5799.5  398.91
#Mann=4,-1,0
  3876.7    0.05       0  4986.0    0.16       0  4987.7    0.07       0
  5007.1    0.16       0
Bank Sta=4987.7,5007.1
Exp/Cntr=0.3,0.1

Type RM Length L Ch R = 1,7620,416,416,416
BEGIN DESCRIPTION:
Mill Creek7619.729
END DESCRIPTION:
XS GIS Cut Line= 3
      2742554.77      6815301.28      2742476.00      6816261.00
      2742401.00      6817036.04
#Sta/Elev= 30
  4041.5  408.96  4071.3  406.90  4087.0  404.70  4131.5  401.73  4262.0  389.18
  4329.6  384.67  4382.4  382.20  4502.8  379.21  4593.1  378.65  4683.4  379.63
  4803.8  379.00  4904.1  380.61  4914.1  380.38  4924.2  374.69  4924.5  372.72
  4925.0  372.22  4943.9  372.72  4946.3  375.72  4955.5  377.41  4984.4  379.81
  5001.9  380.35  5024.5  378.65  5044.6  379.52  5058.0  378.80  5125.0  381.62
  5198.8  383.64  5285.8  386.53  5476.6  391.05  5675.9  398.08  5783.1  401.03
#Mann=5,-1,0
  4041.5    0.05       0  4924.5    0.07       0  4943.9    0.05       0
  4955.5    0.16       0  5198.8    0.05       0
Bank Sta=4924.5,4943.9
Exp/Cntr=0.3,0.1

Type RM Length L Ch R = 1,7204,437,437,437
BEGIN DESCRIPTION:
Mill Creek7204.003
END DESCRIPTION:
XS GIS Cut Line= 3
      2742178.96      6815339.08      2742176.00      6816011.00
      2742176.00      6817110.98
#Sta/Elev= 30
  4324.1  411.59  4426.0  405.27  4496.0  399.44  4536.0  392.12  4606.0  385.85
  4686.0  379.82  4726.0  377.76  4796.0  376.91  4846.0  378.63  4976.0  379.63
  4983.8  372.10  4984.3  371.60  5002.7  371.60  5003.2  372.10  5036.0  378.75
  5046.0  379.17  5066.0  379.81  5106.0  379.67  5136.0  378.75  5215.1  379.22
  5296.0  378.92  5326.0  378.20  5356.0  380.31  5381.8  380.65  5466.0  381.89
  5556.0  384.87  5596.0  385.11  5616.0  386.57  5896.0  394.93  6096.0  402.12
#Mann=5,-1,0
  4324.1    0.05       0  4983.8    0.05       0  5003.2    0.05       0
  5215.1    0.16       0  5381.8    0.05       0
Bank Sta=4983.8,5003.2
Exp/Cntr=0.3,0.1

Type RM Length L Ch R = 1,6767,463,463,463
BEGIN DESCRIPTION:
Mill Creek6767.169
END DESCRIPTION:
XS GIS Cut Line= 3
      2741876.00      6815410.97      2741876.00      6815911.00
      2741676.00      6817111.02
#Sta/Elev= 30
  4503.9  413.56  4523.9  412.22  4533.9  410.52  4553.9  405.53  4613.9  393.96
  4643.9  390.53  4693.9  386.44  4733.9  382.22  4773.9  379.41  4813.9  377.56
  4843.9  377.25  4943.9  378.92  4953.9  377.97  4963.9  374.55  4964.1  371.43
  4964.6  370.93  4983.2  370.93  4983.7  371.43  4983.9  373.97  4993.9  378.43
  5001.4  378.66  5024.2  378.13  5085.0  379.19  5462.7  377.15  5706.0  380.99
  5815.0  385.08  5855.5  387.83  6010.1  395.99  6139.4  400.97  6220.5  402.58
#Mann=3,-1,0
  4503.9    0.05       0  4964.1    0.05       0  4983.7    0.05       0
Bank Sta=4964.1,4983.7
Exp/Cntr=0.3,0.1

Type RM Length L Ch R = 1,6304,308,308,308
BEGIN DESCRIPTION:
Mill Creek6304.35
END DESCRIPTION:
XS GIS Cut Line= 3
      2741432.91      6815112.33      2741430.09      6815971.20
      2741452.89      6817481.86
#Sta/Elev= 30
  4154.2  399.94  4232.9  399.62  4302.9  397.52  4452.9  387.97  4712.9  381.15
  4736.6  380.02  4762.9  376.39  4782.9  375.60  4832.9  375.27  4862.9  377.02
  4892.9  375.16  4962.9  377.76  4972.9  376.75  4982.9  372.49  4983.1  370.69
  4983.6  370.19  5002.7  370.69  5010.5  377.52  5070.7  376.40  5412.9  376.25
  5522.9  379.75  5843.0  384.70  5923.0  388.74  5964.3  392.15  5993.0  394.15
  6043.0  395.38  6223.0  394.48  6393.0  395.41  6403.2  396.32  6523.9  396.11
#Mann=4,-1,0
  4154.2    0.05       0  4983.1    0.05       0  5002.7    0.05       0
  5964.3    0.16       0
Bank Sta=4983.1,5002.7
Exp/Cntr=0.3,0.1

Type RM Length L Ch R = 1,5996,475,475,475
BEGIN DESCRIPTION:
Mill Creek5996.3
END DESCRIPTION:
XS GIS Cut Line= 3
      2741169.90      6815043.70      2741174.61      6815833.49
      2741046.11      6817526.82
#Sta/Elev= 30
  4229.0  390.60  4417.4  386.80  4676.3  378.87  4926.3  376.12  4976.3  377.38
  4986.3  376.81  4986.5  369.86  4987.0  369.36  5006.1  369.86  5026.3  371.31
  5036.4  377.18  5156.7  377.25  5248.9  375.61  5377.3  376.09  5462.8  379.62
  5612.2  378.31  5658.1  378.55  5668.2  377.42  5678.2  378.80  5725.3  377.43
  5938.9  380.66  6099.4  384.15  6124.1  386.39  6255.4  386.66  6340.1  389.82
  6470.5  390.03  6540.7  393.65  6649.1  395.13  6654.2  396.56  6717.0  395.21
#Mann=5,-1,0
  4229.0   0.035       0  4986.5   0.035       0  5006.1   0.035       0
  5248.9    0.07       0  5612.2    0.05       0
Bank Sta=4986.5,5006.1
Exp/Cntr=0.3,0.1

Type RM Length L Ch R = 1,5521,325,325,325
BEGIN DESCRIPTION:
Mill Creek5520.768
END DESCRIPTION:
XS GIS Cut Line= 3
      2740843.39      6814925.06      2740835.14      6815661.11
      2740751.00      6817185.99
#Sta/Elev= 30
  4263.9  399.52  4288.3  396.42  4369.8  387.93  4445.7  382.28  4509.9  379.80
  4777.8  375.89  4789.9  376.35  4829.9  374.54  4875.7  375.09  4969.9  376.57
  4979.9  370.65  4980.1  369.44  4980.6  368.94  4999.7  369.44  5002.4  370.20
  5009.9  375.39  5019.9  376.59  5121.4  374.93  5160.1  375.70  5210.2  373.58
  5267.5  375.27  5365.4  376.14  5450.6  374.74  5493.3  375.38  5709.7  376.17
  5841.2  377.23  6021.4  383.04  6121.6  391.14  6311.9  401.54  6527.2  403.07
#Mann=12,-1,0
  4263.9    0.07       0  4288.3    0.16       0  4445.7    0.12       0
  4777.8   0.035       0  4875.7    0.16       0  4980.1    0.07       0
  4999.7    0.16       0  5121.4    0.12       0  5267.5    0.16       0
  5365.4    0.05       0  5493.3    0.16       0  5709.7    0.05       0
Bank Sta=4980.1,4999.7
Exp/Cntr=0.3,0.1
