--- Persimmon Branch.prj (project) ---

Proj Title=Persimmon Branch Base Level Engineering
Current Plan=p01
Default Exp/Contr=0.3,0.1
English Units
Geom File=g01
Flow File=f01
Plan File=p01
BEGIN DESCRIPTION:
Persimmon Branch
END DESCRIPTION:

--- Persimmon Branch.p01 (plan) ---

Plan Title=Multiple Run
Short Identifier=Multiple
Geom File=g01
Flow File=f01
Subcritical Flow
K Sum by GR= 0
Std Step Tol= 0.01
Critical Tol= 0.01
Num of Std Step Trials= 20
Max Error Tol= 0.3
Flow Tol Ratio= 0.001
Split Flow NTrial= 30
Split Flow Tol= 0.02
Split Flow Ratio= 0.02
Log Output Level= 0
Friction Slope Method= 1
Unsteady Friction Slope Method= 2
Unsteady Bridges Friction Slope Method= 1
Parabolic Critical Depth
Global Vel Dist=  1 , 1 , 1
Global Log Level= 0
CheckData=True
Encroach Param= -1, 0, 0, 0
BEGIN DESCRIPTION:
Multiple Run
END DESCRIPTION:

--- Persimmon Branch.f01 (steady flow) ---

Flow Title=Multiple
Number of Profiles=7
Profile Names=10-year,25-year,50-year,1pct_min,100-year,1pct_plu,500-year
River Rch & RM= Persimmon Branch,Reach-1,24362
     401     525     621     365     729    1455    1003
River Rch & RM= Persimmon Branch,Reach-1,22512
     666     895    1079     645    1288    2569    1832
River Rch & RM= Persimmon Branch,Reach-1,17431
     974    1334    1630     986    1966    3923    2864
River Rch & RM= Persimmon Branch,Reach-1,13466
    1021    1402    1715    1039    2072    4134    3026
River Rch & RM= Persimmon Branch,Reach-1,12740
    1516    2121    2628    1609    3210    6404    4794
River Rch & RM= Persimmon Branch,Reach-1,9718
    1706    2398    2981    1830    3652    7286    5486
River Rch & RM= Persimmon Branch,Reach-1,7716
    1699    2379    2949    1805    3602    7186    5378
River Rch & RM= Persimmon Branch,Reach-1,4299
    1861    2607    3232    1977    3946    7872    5886
River Rch & RM= Persimmon Branch,Reach-1,3038
    1942    2717    3366    2057    4104    8188    6108
Boundary for River Rch & Prof#=Persimmon Branch,Reach-1,1
Up Type=0
Dn Type=3
Dn Slope=0.005
Boundary for River Rch & Prof#=Persimmon Branch,Reach-1,2
Up Type=0
Dn Type=3
Dn Slope=0.005
Boundary for River Rch & Prof#=Persimmon Branch,Reach-1,3
Up Type=0
Dn Type=3
Dn Slope=0.005
Boundary for River Rch & Prof#=Persimmon Branch,Reach-1,4
Up Type=0
Dn Type=3
Dn Slope=0.005
Boundary for River Rch & Prof#=Persimmon Branch,Reach-1,5
Up Type=0
Dn Type=3
Dn Slope=0.005
Boundary for River Rch & Prof#=Persimmon Branch,Reach-1,6
Up Type=0
Dn Type=3
Dn Slope=0.005
Boundary for River Rch & Prof#=Persimmon Branch,Reach-1,7
Up Type=0
Dn Type=3
Dn Slope=0.005

--- Persimmon Branch.g01 (geometry) ---

Geom Title=Existing Conditions

River Reach=Persimmon Branch,Reach-1
Reach XY= 30
      2667776.00      6819761.00      2667835.41      6820417.62
      2668437.53      6821259.50      2669605.57      6821461.53
      2672826.31      6821503.77      2672927.28      6821364.38
      2673310.59      6821460.98      2673532.06      6821352.86
      2673722.46      6821159.54      2673733.69      6820854.52
      2674618.26      6819817.46      2674636.34      6819450.88
      2674870.96      6819355.92      2675131.44      6818866.25
      2675426.00      6818761.00      2675379.18      6818262.41
      2675773.18      6817953.05      2675729.04      6817762.42
      2676381.26      6816316.47      2677023.05      6815609.00
      2676945.17      6815491.03      2677517.03      6815067.67
      2677581.83      6814608.69      2677825.48      6814495.45
      2677731.30      6814108.46      2678206.37      6813881.68
      2678466.20      6813371.48      2679885.62      6812462.27
      2682520.56      6812358.84      2683726.00      6811311.00

Type RM Length L Ch R = 1,24362,461,461,461
BEGIN DESCRIPTION:
Persimmon Branch 35
END DESCRIPTION:
XS GIS Cut Line= 3
      2666875.98      6820111.01      2667776.00      6819911.00
      2668326.00      6820011.00
#Sta/Elev= 30
  4084.6  389.39  4166.6  387.72  4217.8  385.09  4320.2  383.81  4330.5  383.56
  4336.9  382.79  4443.2  380.35  4521.3  377.84  4627.6  377.65  4699.3  375.57
  4797.9  374.84  4904.1  375.50  5004.0  374.15  5026.9  374.49  5098.1  374.05
  5128.5  374.57  5148.1  373.11  5148.4  372.61  5151.9  372.61  5152.1  373.11
  5169.2  375.14  5203.5  374.48  5256.9  376.72  5352.2  377.85  5403.0  379.15
  5422.0  380.24  5427.1  379.92  5504.6  381.79  5514.8  383.02  5565.6  385.11
#Mann=3,-1,0
  4084.6    0.05       0  5148.1    0.04       0  5152.1    0.05       0
Bank Sta=5148.1,5152.1
Exp/Cntr=0.3,0.1

Type RM Length L Ch R = 1,23901,476,476,476
BEGIN DESCRIPTION:
Persimmon Branch 34
END DESCRIPTION:
XS GIS Cut Line= 3
      2667026.04      6820460.99      2667876.00      6820311.00
      2668326.02      6820060.99
#Sta/Elev= 30
  4138.0  387.57  4371.5  382.44  4523.8  376.03  4544.1  378.15  4564.4  379.11
  4623.7  378.94  4628.8  375.96  4655.8  378.83  4666.0  378.77  4682.9  375.94
  4688.0  376.55  4696.5  374.12  4706.6  373.92  4767.5  374.45  4855.5  372.81
  5004.0  372.85  5024.0  372.59  5030.8  371.53  5066.6  371.35  5066.8  370.85
  5070.6  371.35  5074.3  372.02  5090.3  371.46  5096.0  372.30  5112.1  371.36
  5161.2  373.79  5404.9  379.97  5435.8  381.26  5458.7  383.30  5515.9  385.37
#Mann=3,-1,0
  4138.0    0.05       0  5066.6    0.04       0  5070.6    0.05       0
Bank Sta=5066.6,5070.6
Exp/Cntr=0.3,0.1

Type RM Length L Ch R = 1,23425,203,203,203
BEGIN DESCRIPTION:
Persimmon Branch 349
END DESCRIPTION:
XS GIS Cut Line= 3
      2667231.48      6820834.07      2668027.93      6820705.78
      2668601.30      6820276.81
#Sta/Elev= 30
  4189.3  380.68  4224.3  380.00  4234.4  379.46  4244.8  377.29  4301.6  375.00
  4396.5  373.66  4406.6  372.85  4568.6  371.66  4842.1  370.94  4882.6  371.38
  4913.0  370.66  4991.8  370.36  5004.1  368.50  5004.3  368.00  5007.8  368.00
  5008.1  368.50  5041.5  370.31  5127.0  371.04  5177.0  372.52  5277.0  372.85
  5341.6  374.76  5347.9  375.59  5377.1  375.33  5447.9  378.30  5462.5  380.01
  5483.3  379.83  5533.3  380.96  5555.6  382.69  5583.4  383.77  5712.1  384.96
#Mann=3,-1,0
  4189.3    0.05       0  5004.1    0.04       0  5008.1    0.05       0
Bank Sta=5004.1,5008.1
Exp/Cntr=0.3,0.1

Type RM Length L Ch R = 1,23222,334,334,334
BEGIN DESCRIPTION:
Persimmon Branch 348
END DESCRIPTION:
XS GIS Cut Line= 3
      2667308.12      6821163.03      2668170.91      6820823.15
      2668671.60      6820481.10
#Sta/Elev= 30
  4060.0  376.71  4090.0  376.99  4106.3  375.76  4111.6  376.59  4130.7  374.71
  4136.0  376.09  4160.4  372.65  4165.8  373.82  4184.8  371.63  4214.6  371.25
  4390.9  370.79  4406.8  371.95  4461.0  370.41  4466.3  371.37  4485.4  370.55
  4490.7  371.45  4569.3  371.39  4574.6  370.18  4593.7  370.89  4677.6  369.34
  4929.3  368.80  4987.3  369.66  5018.7  368.51  5019.0  368.01  5022.7  368.51
  5272.0  373.45  5358.7  376.99  5460.3  378.71  5481.3  380.10  5593.7  381.13
#Mann=3,-1,0
  4060.0    0.05       0  5018.7    0.04       0  5022.7    0.05       0
Bank Sta=5018.7,5022.7
Exp/Cntr=0.3,0.1

Type RM Length L Ch R = 1,22888,376,376,376
BEGIN DESCRIPTION:
Persimmon Branch 347
END DESCRIPTION:
XS GIS Cut Line= 3
      2667096.81      6821350.69      2668264.44      6821188.83
      2668711.97      6820633.52
#Sta/Elev= 30
  3653.4  373.73  3773.7  372.45  4005.9  371.14  4016.0  371.51  4026.1  370.94
  4051.5  370.52  4096.8  370.81  4238.1  369.61  4266.8  369.95  4271.8  369.51
  4409.8  369.61  4500.6  368.86  4692.4  368.77  4839.2  367.87  4917.6  368.36
  4938.4  367.74  4971.6  367.60  4971.9  367.10  4975.4  367.10  4975.6  367.60
  5023.2  369.36  5137.6  370.25  5194.3  371.25  5208.7  371.88  5279.1  372.57
  5386.3  374.43  5443.8  376.00  5499.9  376.70  5522.2  377.54  5545.4  377.59
#Mann=3,-1,0
  3653.4    0.05       0  4971.6    0.04       0  4975.6    0.05       0
Bank Sta=4971.6,4975.6
Exp/Cntr=0.3,0.1

Type RM Length L Ch R = 1,22512,375,375,375
BEGIN DESCRIPTION:
Persimmon Branch 346
END DESCRIPTION:
XS GIS Cut Line= 3
      2667532.82      6822196.47      2668505.32      6821469.37
      2668867.77      6820594.97
#Sta/Elev= 30
  3561.1  378.16  3710.4  372.58  3810.5  370.66  3966.8  369.50  3975.1  367.91
  3989.6  367.34  4367.0  367.07  4644.2  365.46  4644.5  364.96  4648.2  365.46
  4675.4  365.68  4681.7  367.09  4688.8  367.39  4696.3  367.14  4702.5  365.78
  4717.1  367.02  4725.5  366.57  4731.7  367.56  4795.4  366.44  4860.2  367.77
  4881.8  366.70  4920.3  367.56  4990.1  366.03  5011.7  366.85  5026.6  366.40
  5050.5  367.92  5163.3  367.70  5417.3  370.80  5465.1  372.38  5721.9  375.87
#Mann=3,-1,0
  3561.1    0.05       0  4644.2    0.04       0  4648.2    0.05       0
Bank Sta=4644.2,4648.2
Exp/Cntr=0.3,0.1

Type RM Length L Ch R = 1,22137,776,776,776
BEGIN DESCRIPTION:
Persimmon Branch 345
END DESCRIPTION:
XS GIS Cut Line= 3
      2667929.00      6822636.19      2668954.16      6821307.62
      2669041.02      6820551.31
#Sta/Elev= 30
  3326.6  366.95  3399.0  366.39  3428.0  367.65  3498.6  366.40  3691.6  364.90
  4262.2  365.39  4561.1  364.20  4697.3  365.62  4718.8  366.68  4725.1  366.49
  4733.3  363.84  4739.6  363.98  4747.8  365.91  4754.0  364.38  4760.5  363.81
  4768.6  364.68  4789.4  364.85  4801.9  363.58  4802.1  363.08  4805.9  363.58
  4811.0  364.90  4818.4  365.36  4889.0  364.33  4938.8  364.81  5004.7  363.96
  5273.1  366.01  5590.3  370.91  5625.4  370.80  5695.8  373.24  5766.0  374.01
#Mann=3,-1,0
  3326.6    0.05       0  4801.9    0.04       0  4805.9    0.05       0
Bank Sta=4801.9,4805.9
Exp/Cntr=0.3,0.1

Type RM Length L Ch R = 1,21361,659,659,659
BEGIN DESCRIPTION:
Persimmon Branch 3420
END DESCRIPTION:
XS GIS Cut Line= 3
      2667909.77      6822857.71      2669623.82      6821481.67
      2669558.48      6820634.74
#Sta/Elev= 30
  2781.7  365.76  2926.3  363.97  3132.7  363.13  3295.9  364.00  3644.7  363.14
  3764.8  363.55  4014.4  362.65  4277.2  363.57  4832.1  361.54  4846.5  361.99
  4887.7  361.08  4887.9  360.58  4891.4  360.58  4891.7  361.08  4896.1  362.19
  4904.1  362.42  4924.9  361.56  4968.1  361.33  4974.5  362.76  4990.5  361.67
  5040.6  361.31  5361.6  361.67  5612.3  363.25  5666.9  363.95  5692.5  365.87
  5712.6  368.71  5722.6  369.18  5752.7  365.91  5762.7  366.47  5829.2  366.53
#Mann=3,-1,0
  2781.7    0.05       0  4887.7    0.04       0  4891.7    0.05       0
Bank Sta=4887.7,4891.7
Exp/Cntr=0.3,0.1

Type RM Length L Ch R = 1,20702,699,699,699
BEGIN DESCRIPTION:
Persimmon Branch 3419
END DESCRIPTION:
XS GIS Cut Line= 3
      2668030.59      6822979.81      2670250.34      6821464.05
      2669930.52      6820372.96
#Sta/Elev= 30
  2309.1  363.33  2384.5  362.20  2549.1  362.63  2578.9  361.96  2902.0  362.34
  3003.6  361.76  3045.6  362.73  3096.4  362.18  4773.8  359.81  4816.2  360.19
  4822.2  360.80  4831.1  360.31  4844.0  357.71  4844.3  357.21  4847.8  357.21
  4848.0  357.71  4852.1  360.20  4873.1  360.46  4902.9  359.86  4917.8  358.65
  4931.2  359.13  4938.8  358.32  4944.9  359.65  4959.8  360.06  4974.7  358.48
  4980.8  359.43  4995.3  360.05  5656.7  360.54  5969.3  362.01  6134.0  363.92
#Mann=3,-1,0
  2309.1    0.05       0  4844.0    0.03       0  4848.0    0.05       0
Bank Sta=4844,4848
Exp/Cntr=0.3,0.1

Type RM Length L Ch R = 1,20003,478,478,478
BEGIN DESCRIPTION:
Persimmon Branch 3421
END DESCRIPTION:
XS GIS Cut Line= 3
      2668868.20      6823392.75      2670967.85      6821521.14
      2670567.95      6820245.48
#Sta/Elev= 30
  2071.5  358.42  3239.8  358.79  3289.1  359.69  4104.3  358.66  4125.2  359.42
  4167.8  358.15  4855.0  357.26  4936.0  356.23  4968.2  357.30  4973.7  354.40
  4977.0  353.78  4977.2  353.28  4981.0  353.78  4989.2  357.14  4999.6  357.65
  5031.1  357.03  5356.0  357.56  5366.4  357.01  5460.8  357.78  5481.7  357.22
  5722.8  357.91  5984.8  359.54  6107.9  361.34  6113.2  362.73  6140.4  362.32
  6145.6  363.68  6172.8  363.17  6178.1  364.38  6204.8  364.03  6221.1  364.73
#Mann=3,-1,0
  2071.5    0.05       0  4977.0    0.03       0  4981.0    0.05       0
Bank Sta=4977,4981
Exp/Cntr=0.3,0.1

Type RM Length L Ch R = 1,19525,278,278,278
BEGIN DESCRIPTION:
Persimmon Branch 3422
END DESCRIPTION:
XS GIS Cut Line= 3
      2669326.66      6823397.46      2671396.60      6821473.29
      2671318.84      6819975.75
#Sta/Elev= 30
  2161.7  357.66  2547.8  357.33  2965.6  358.36  3120.9  357.67  3326.2  358.43
  3347.7  357.81  3389.7  358.66  3609.1  358.28  3616.4  359.11  3673.1  357.87
  3899.3  358.11  4663.5  355.93  4939.5  356.16  5010.2  355.84  5028.2  353.49
  5028.4  352.99  5031.9  352.99  5032.2  353.49  5040.2  355.89  5095.6  355.27
  5100.6  355.77  5160.4  355.41  5390.7  356.51  5560.9  356.03  5771.2  356.78
  5781.2  356.16  5841.3  356.71  6021.5  356.52  6412.0  357.35  6487.4  358.20
#Mann=3,-1,0
  2161.7    0.05       0  5028.2    0.03       0  5032.2    0.05       0
Bank Sta=5028.2,5032.2
Exp/Cntr=0.3,0.1

Type RM Length L Ch R = 1,19247,508,508,508
BEGIN DESCRIPTION:
Persimmon Branch 3423
END DESCRIPTION:
XS GIS Cut Line= 3
      2669476.19      6823416.25      2671660.95      6821686.82
      2671549.58      6819914.43
#Sta/Elev= 30
  1987.6  357.47  2567.8  357.87  2588.6  357.25  2603.1  357.81  2944.4  357.54
  3066.3  356.80  3159.2  357.98  3194.5  357.23  3535.8  357.70  4120.4  356.09
  4246.4  355.47  4660.9  354.55  4681.7  355.50  4710.6  354.44  4819.9  354.36
  4960.2  354.43  5010.3  355.30  5018.3  351.98  5018.6  351.48  5022.3  351.98
  5030.3  354.75  5040.4  355.20  5290.8  355.28  5408.5  356.32  5761.8  355.46
  5771.8  354.34  5801.9  355.25  6012.3  356.34  6112.5  356.10  6549.9  358.17
#Mann=5,-1,0
  1987.6    0.05       0  4120.4    0.12       0  4246.4    0.05       0
  5018.3    0.03       0  5022.3    0.05       0
Bank Sta=5018.3,5022.3
Exp/Cntr=0.3,0.1

Type RM Length L Ch R = 1,18739,553,553,553
BEGIN DESCRIPTION:
Persimmon Branch 3418
END DESCRIPTION:
XS GIS Cut Line= 3
      2670358.35      6823419.68      2672172.43      6821441.24
      2671652.20      6819826.82
#Sta/Elev= 30
  2342.9  355.51  2375.7  356.67  3373.4  355.27  3423.3  355.96  3812.4  355.68
  4067.1  354.65  4145.4  355.53  4251.5  354.18  4994.5  353.94  5020.8  350.96
  5021.1  350.46  5024.8  350.96  5032.2  350.96  5037.9  354.17  5048.4  353.17
  5395.4  354.03  5563.2  353.29  5684.0  353.85  5741.8  353.11  6298.4  355.82
  6330.2  356.78  6361.7  356.52  6373.0  357.73  6393.2  356.77  6414.2  357.90
  6431.9  357.26  6437.1  358.17  6456.2  357.05  6487.8  356.82  6723.3  358.42
#Mann=3,-1,0
  2342.9    0.05       0  5020.8    0.03       0  5024.8    0.05       0
Bank Sta=5020.8,5024.8
Exp/Cntr=0.3,0.1

Type RM Length L Ch R = 1,18186,352,352,352
BEGIN DESCRIPTION:
Persimmon Branch 337
END DESCRIPTION:
XS GIS Cut Line= 3
      2672638.26      6823034.26      2672707.46      6821472.03
      2672680.29      6820489.57
#Sta/Elev= 30
  3425.4  353.87  3989.2  352.94  4029.3  354.41  4059.3  352.99  4159.4  351.84
  4549.8  351.37  4559.8  352.35  4579.8  351.41  4589.8  352.21  4860.1  352.81
  4890.1  351.80  4992.2  352.12  5000.2  351.62  5008.2  348.46  5008.4  347.96
  5012.2  348.46  5020.2  351.25  5030.2  352.55  5050.2  350.80  5100.2  351.04
  5200.3  349.71  5400.3  351.97  5430.4  351.06  5460.4  352.29  5630.4  352.24
  5720.5  353.38  5730.5  352.48  5830.5  353.91  5860.5  353.18  5972.0  353.87
#Mann=3,-1,0
  3425.4    0.05       0  5008.2    0.03       0  5012.2    0.05       0
Bank Sta=5008.2,5012.2
Exp/Cntr=0.3,0.1

Type RM Length L Ch R = 1,17834,403,403,403
BEGIN DESCRIPTION:
Persimmon Branch 333
END DESCRIPTION:
XS GIS Cut Line= 3
      2672934.67      6822988.75      2672965.34      6821373.72
      2673010.58      6820305.29
#Sta/Elev= 30
  3371.6  353.29  3419.4  353.83  3439.4  353.36  3669.4  353.23  4149.5  351.60
  4469.5  349.43  4539.6  349.56  4589.6  351.03  4709.6  351.11  4789.6  350.56
  4829.6  351.11  4939.6  349.76  5009.7  349.86  5027.5  348.68  5027.9  348.18
  5031.5  348.18  5031.9  348.68  5039.7  349.48  5109.7  350.61  5122.7  351.23
  5179.8  350.77  5356.0  351.74  5370.0  351.36  5630.2  352.00  5640.2  352.54
  5690.3  352.97  5790.4  352.64  5820.4  353.56  5950.5  352.79  6056.3  353.21
#Mann=3,-1,0
  3371.6    0.05       0  5027.5    0.04       0  5031.9    0.05       0
Bank Sta=5027.5,5031.9
Exp/Cntr=0.3,0.1

Type RM Length L Ch R = 1,17431,479,479,479
BEGIN DESCRIPTION:
Persimmon Branch 334
END DESCRIPTION:
XS GIS Cut Line= 3
      2673523.88      6822658.71      2673307.09      6821474.66
      2673101.59      6820379.20
#Sta/Elev= 30
  3782.2  352.70  4389.8  352.14  4603.3  351.47  4623.7  351.01  4664.3  351.78
  4755.8  351.05  4766.0  351.52  4799.6  351.48  4827.0  350.38  4847.3  350.33
  4877.8  349.20  4911.1  349.09  4949.0  347.87  5060.9  348.53  5072.3  347.72
  5072.8  347.22  5076.5  347.22  5077.1  347.72  5091.4  348.68  5152.4  348.13
  5172.8  349.24  5203.3  349.65  5213.5  350.24  5232.3  349.21  5305.1  350.26
  5457.8  350.72  5505.3  350.00  5640.8  351.16  5691.7  350.99  6100.5  352.64
#Mann=3,-1,0
  3782.2    0.05       0  5072.3    0.04       0  5077.1    0.05       0
Bank Sta=5072.3,5077.1
Exp/Cntr=0.3,0.1

Type RM Length L Ch R = 1,16952,609,609,609
BEGIN DESCRIPTION:
Persimmon Branch 335
END DESCRIPTION:
XS GIS Cut Line= 3
      2674276.28      6822124.37      2673696.40      6821212.98
      2673134.84      6820270.88
#Sta/Elev= 30
  3902.8  352.81  4049.0  352.39  4064.2  353.02  4085.4  352.32  4158.2  351.88
  4173.5  352.48  4209.9  351.86  4274.2  352.07  4303.8  351.37  4470.6  351.02
  4528.2  350.48  4564.6  349.47  4665.4  348.78  4846.6  348.57  4890.6  347.73
  4961.7  347.94  4992.4  347.07  5013.8  347.66  5109.2  347.75  5186.6  346.79
  5187.1  346.29  5190.8  346.29  5191.4  346.79  5342.8  347.59  5502.4  349.53
  5518.0  349.13  5730.2  351.02  5831.4  350.94  5932.6  352.15  6079.8  352.45
#Mann=3,-1,0
  3902.8    0.05       0  5186.6    0.04       0  5191.4    0.05       0
Bank Sta=5186.6,5191.4
Exp/Cntr=0.3,0.1

Type RM Length L Ch R = 1,16343,541,541,541
BEGIN DESCRIPTION:
Persimmon Branch 336
END DESCRIPTION:
XS GIS Cut Line= 3
      2674558.56      6821714.89      2673940.73      6820724.75
      2673360.79      6820026.59
#Sta/Elev= 30
  3812.6  352.44  3840.3  352.70  3946.8  352.06  4019.6  351.95  4077.4  352.34
  4194.4  351.70  4370.0  351.69  4601.2  350.41  4653.1  350.52  4789.9  349.43
  4884.3  348.06  4890.2  347.58  4899.7  348.13  4957.5  345.97  4993.0  345.48
  4999.5  345.22  5011.2  342.61  5011.9  342.11  5015.7  342.11  5016.5  342.61
  5021.6  343.84  5028.1  344.63  5042.5  345.54  5163.6  346.45  5241.7  347.86
  5433.1  350.18  5638.8  351.18  5731.3  351.84  5802.9  352.92  5887.3  353.28
#Mann=3,-1,0
  3812.6    0.05       0  5011.2    0.03       0  5016.5    0.05       0
Bank Sta=5011.2,5016.5
Exp/Cntr=0.3,0.1

Type RM Length L Ch R = 1,15802,504,504,504
BEGIN DESCRIPTION:
Persimmon Branch 332
END DESCRIPTION:
XS GIS Cut Line= 3
      2674881.44      6820860.41      2674279.06      6820306.98
      2673642.82      6819960.66
#Sta/Elev= 30
  4174.9  352.08  4235.2  352.32  4249.4  351.57  4426.3  351.29  4440.3  351.74
  4447.3  350.91  4645.2  350.19  4673.6  349.44  4744.5  349.10  4772.8  348.03
  4815.4  347.95  4987.0  344.37  5007.8  344.24  5017.6  340.85  5018.4  340.35
  5023.1  340.85  5030.6  343.06  5036.5  344.02  5080.2  345.42  5099.1  344.85
  5155.8  346.05  5227.4  345.98  5347.1  347.36  5368.9  348.20  5412.6  348.47
  5440.4  349.68  5603.5  350.70  5656.8  351.47  5679.5  353.00  5717.3  352.48
#Mann=5,-1,0
  4174.9    0.05       0  4987.0    0.12       0  5017.6    0.07       0
  5023.1    0.12       0  5099.1    0.05       0
Bank Sta=5017.6,5023.1
Exp/Cntr=0.3,0.1

Type RM Length L Ch R = 1,15298,213,213,213
BEGIN DESCRIPTION:
Persimmon Branch 331
END DESCRIPTION:
XS GIS Cut Line= 3
      2675419.16      6819975.31      2674527.31      6819902.12
      2673655.72      6819891.64
#Sta/Elev= 30
  4101.5  350.48  4295.3  349.32  4334.0  348.84  4339.0  348.04  4365.5  348.75
  4496.0  347.83  4506.0  349.17  4626.4  346.79  4646.5  347.45  4867.2  344.99
  4937.5  343.27  4967.6  343.43  4977.6  339.87  4984.8  338.94  4985.7  338.44
  4990.4  338.94  4999.5  339.65  5007.7  343.21  5017.7  343.94  5117.7  344.17
  5230.3  345.76  5329.3  347.06  5407.7  348.93  5487.7  349.85  5509.1  349.27
  5657.7  351.85  5677.7  351.22  5767.7  351.83  5817.7  353.18  5868.0  352.72
#Mann=5,-1,0
  4101.5    0.05       0  4984.8    0.03       0  4990.4    0.05       0
  5230.3    0.12       0  5329.3    0.05       0
Bank Sta=4984.8,4990.4
Exp/Cntr=0.3,0.1

Type RM Length L Ch R = 1,15085,323,323,323
BEGIN DESCRIPTION:
Persimmon Branch 330
END DESCRIPTION:
XS GIS Cut Line= 3
      2675438.22      6819760.69      2674626.78      6819745.84
      2673592.00      6819621.47
#Sta/Elev= 30
  4188.0  348.84  4620.3  347.83  4660.3  347.00  4760.3  346.68  4880.3  344.31
  4970.4  343.96  4980.4  343.26  4988.0  341.68  4993.0  341.59  5020.5  342.23
  5040.7  343.52  5057.8  339.26  5058.8  338.76  5062.8  338.76  5063.8  339.26
  5070.9  343.02  5079.0  344.09  5101.1  343.38  5166.2  343.43  5191.7  344.00
  5221.9  345.85  5262.2  346.33  5317.9  347.37  5363.0  348.65  5383.1  348.07
  5423.4  349.45  5645.0  352.14  5725.5  352.55  5997.5  355.73  6041.8  355.50
#Mann=5,-1,0
  4188.0    0.05       0  5057.8    0.03       0  5063.8    0.05       0
  5262.2    0.12       0  5317.9    0.05       0
Bank Sta=5057.8,5063.8
Exp/Cntr=0.3,0.1

Type RM Length L Ch R = 1,14762,500,500,500
BEGIN DESCRIPTION:
Persimmon Branch 329
END DESCRIPTION:
XS GIS Cut Line= 3
      2675452.89      6819749.70      2674796.35      6819568.45
      2674225.58      6819025.01
#Sta/Elev= 30
  4123.1  348.82  4462.2  347.33  4483.0  347.89  4493.3  347.06  4597.1  346.06
  4663.8  347.01  4703.3  345.52  4731.9  345.66  4752.7  344.55  4880.4  342.05
  4937.1  342.87  4944.0  341.86  4951.2  342.93  4972.8  343.52  4986.4  342.98
  5000.6  343.73  5007.8  339.69  5014.7  338.90  5022.0  341.05  5028.9  340.91
  5036.2  342.46  5057.2  342.06  5061.4  338.90  5062.5  338.40  5067.5  338.90
  5078.6  342.43  5097.6  343.63  5248.1  345.32  5340.3  347.66  5592.3  351.46
#Mann=5,-1,0
  4123.1    0.05       0  4972.8    0.12       0  5061.4    0.07       0
  5067.5    0.12       0  5097.6    0.05       0
Bank Sta=5061.4,5067.5
Exp/Cntr=0.3,0.1

Type RM Length L Ch R = 1,14262,270,270,270
BEGIN DESCRIPTION:
Persimmon Branch 328
END DESCRIPTION:
XS GIS Cut Line= 3
      2675465.18      6819735.82      2674961.99      6819130.67
      2674653.48      6818739.13
#Sta/Elev= 30
  4209.6  348.69  4389.8  347.97  4560.4  346.43  4617.7  346.59  4659.3  345.23
  4702.3  345.26  4844.2  341.95  4896.9  341.51  4908.0  341.70  4944.2  340.76
  4971.8  341.48  4979.6  335.69  4983.1  335.69  4984.1  335.19  4988.2  335.19
  4989.2  335.69  4993.2  339.39  4996.6  339.39  5000.4  337.96  5008.5  341.59
  5014.8  341.98  5050.1  340.57  5136.2  340.07  5172.0  340.49  5240.1  342.84
  5292.2  345.19  5385.3  347.50  5406.1  348.66  5449.4  349.00  5495.1  350.12
#Mann=5,-1,0
  4209.6    0.05       0  4896.9    0.12       0  4983.1    0.07       0
  4989.2    0.12       0  5240.1    0.05       0
Bank Sta=4983.1,4989.2
Exp/Cntr=0.3,0.1

Type RM Length L Ch R = 1,13992,217,217,217
BEGIN DESCRIPTION:
Persimmon Branch 327
END DESCRIPTION:
XS GIS Cut Line= 3
      2675492.47      6819693.92      2675110.22      6818941.50
      2674672.02      6818660.33
#Sta/Elev= 30
  4144.5  348.74  4360.9  347.16  4456.5  345.27  4501.0  345.22  4529.1  344.15
  4540.0  344.29  4551.6  345.45  4612.3  344.93  4629.0  344.20  4679.1  344.29
  4731.0  342.58  4812.6  340.84  4840.5  340.82  4873.8  341.66  4888.1  340.89
  4923.9  341.30  4993.5  340.44  4999.0  339.87  5014.2  340.72  5020.2  338.03
  5038.3  335.24  5039.3  334.74  5044.4  335.24  5050.6  335.82  5056.5  340.72
  5100.4  339.59  5338.3  347.31  5353.2  347.37  5389.5  348.95  5509.1  349.57
#Mann=5,-1,0
  4144.5    0.05       0  4840.5    0.12       0  5038.3    0.07       0
  5044.4    0.12       0  5338.3    0.05       0
Bank Sta=5038.3,5044.4
Exp/Cntr=0.3,0.1

Type RM Length L Ch R = 1,13775,309,309,309
BEGIN DESCRIPTION:
Persimmon Branch 319
END DESCRIPTION:
XS GIS Cut Line= 4
      2675519.52      6819666.28      2675403.08      6819058.23
      2675261.58      6818828.79      2674846.53      6818698.09
#Sta/Elev= 30
  4108.7  348.87  4318.1  347.14  4365.1  345.70  4417.1  346.74  4474.3  345.12
  4501.0  345.55  4643.5  343.23  4682.4  343.52  4687.5  344.19  4737.0  343.67
  4759.8  342.40  4885.4  339.97  4941.6  340.25  4971.3  339.46  4984.2  339.96
  4993.1  334.56  4999.3  334.27  5000.3  333.77  5005.4  334.27  5007.6  338.20
  5013.7  339.64  5024.2  340.15  5034.7  340.20  5045.2  339.06  5072.3  339.74
  5137.0  339.23  5191.9  340.02  5244.6  341.32  5336.5  345.13  5432.5  347.73
#Mann=4,-1,0
  4108.7    0.05       0  4885.4    0.12       0  4999.3    0.07       0
  5005.4    0.12       0
Bank Sta=4999.3,5005.4
Exp/Cntr=0.3,0.1

Type RM Length L Ch R = 1,13466,385,385,385
BEGIN DESCRIPTION:
Persimmon Branch 236
END DESCRIPTION:
XS GIS Cut Line= 3
      2676076.91      6818642.14      2675359.85      6818661.14
      2674782.78      6818665.88
#Sta/Elev= 30
  4298.0  349.71  4338.9  349.92  4388.9  347.99  4499.0  346.25  4529.0  344.85
  4569.0  345.31  4679.0  342.42  4689.0  342.81  4734.1  342.02  4789.1  341.12
  4849.1  341.93  4859.1  340.44  4909.1  338.66  4989.2  338.75  4999.2  337.71
  5005.9  333.27  5007.0  332.77  5012.4  333.27  5014.7  338.94  5089.2  337.52
  5119.2  338.75  5209.2  338.98  5259.2  341.29  5319.2  342.55  5369.2  345.45
  5389.2  345.14  5419.2  345.89  5489.2  348.47  5557.3  348.73  5592.4  348.57
#Mann=5,-1,0
  4298.0    0.05       0  4734.1    0.12       0  5005.9    0.07       0
  5012.4    0.12       0  5557.3    0.05       0
Bank Sta=5005.9,5012.4
Exp/Cntr=0.3,0.1

Type RM Length L Ch R = 1,13081,341,341,341
BEGIN DESCRIPTION:
Persimmon Branch 235
END DESCRIPTION:
XS GIS Cut Line= 3
      2676136.64      6818426.97      2675385.10      6818345.65
      2674729.47      6818655.28
#Sta/Elev= 30
  4235.0  350.51  4346.3  350.32  4537.4  343.86  4619.4  339.96  4638.0  340.61
  4728.5  338.66  4748.6  339.88  4769.3  339.47  4829.1  337.77  5010.8  338.23
  5023.1  337.72  5033.6  334.26  5035.9  332.56  5036.9  332.06  5042.4  332.56
  5045.2  332.73  5056.3  336.98  5078.4  338.22  5090.2  337.41  5135.7  337.92
  5153.0  339.01  5249.6  341.05  5272.4  342.33  5332.8  343.30  5340.7  344.31
  5369.0  344.00  5409.0  346.05  5488.3  347.83  5616.8  348.12  5716.0  349.25
#Mann=5,-1,0
  4235.0    0.05       0  4769.3    0.12       0  5035.9    0.07       0
  5042.4    0.12       0  5616.8    0.05       0
Bank Sta=5035.9,5042.4
Exp/Cntr=0.3,0.1

Type RM Length L Ch R = 1,12740,708,708,708
BEGIN DESCRIPTION:
Persimmon Branch 232
END DESCRIPTION:
XS GIS Cut Line= 3
      2676158.95      6818348.66      2675570.21      6818114.17
      2674911.85      6817431.40
#Sta/Elev= 30
  4365.7  350.73  4487.3  350.32  4498.0  349.89  4505.7  347.58  4511.1  348.59
  4521.1  347.40  4535.4  349.04  4589.3  347.59  4799.4  338.28  5005.1  336.11
  5013.7  330.46  5015.1  329.96  5023.6  330.46  5025.9  331.20  5032.8  336.67
  5146.0  337.24  5195.7  335.10  5301.7  337.81  5386.6  338.32  5393.5  337.52
  5407.6  338.68  5464.2  338.24  5537.3  339.57  5634.0  341.03  5718.9  344.30
  5818.0  346.05  5824.9  347.52  5832.1  346.31  5839.1  347.77  5947.9  350.02
#Mann=5,-1,0
  4365.7    0.05       0  4521.1    0.12       0  5013.7    0.07       0
  5023.6    0.12       0  5537.3    0.05       0
Bank Sta=5013.7,5023.6
Exp/Cntr=0.3,0.1

Type RM Length L Ch R = 1,12032,444,444,444
BEGIN DESCRIPTION:
Persimmon Branch 234
END DESCRIPTION:
XS GIS Cut Line= 3
      2676448.88      6817998.28      2675868.23      6817660.03
      2674979.21      6817257.00
#Sta/Elev= 30
  4331.4  351.08  4412.7  350.73  4440.0  349.10  4705.1  344.86  4872.6  337.90
  4891.7  335.66  4901.8  332.70  4904.8  329.31  4906.2  328.81  4914.8  329.31
  4925.0  329.68  4931.3  334.02  4937.1  332.29  4947.1  334.67  4952.8  332.80
  4959.7  334.60  4990.1  335.10  5063.9  334.08  5104.6  335.00  5138.7  333.94
  5192.5  335.02  5259.6  334.56  5277.2  335.71  5291.3  334.71  5448.1  337.82
  5542.2  340.31  5622.4  344.14  5910.5  350.41  5928.1  352.62  5979.5  352.91
#Mann=5,-1,0
  4331.4    0.05       0  4891.7    0.12       0  4904.8    0.07       0
  4914.8    0.12       0  5448.1    0.05       0
Bank Sta=4904.8,4914.8
Exp/Cntr=0.3,0.1

Type RM Length L Ch R = 1,11588,262,262,262
BEGIN DESCRIPTION:
Persimmon Branch 233
END DESCRIPTION:
XS GIS Cut Line= 3
      2676473.48      6817274.94      2675985.79      6817257.38
      2675019.29      6817170.63
#Sta/Elev= 30
  4509.9  350.48  4567.4  348.65  4597.4  349.83  4707.5  346.36  4777.6  342.36
  4901.4  337.72  4917.6  336.37  4947.7  330.87  4957.7  331.92  4977.7  331.80
  4982.6  328.48  4984.0  327.98  4992.8  328.48  5000.3  329.18  5013.0  333.42
  5098.1  334.03  5129.2  330.91  5178.4  331.91  5188.5  335.18  5240.3  334.34
  5263.9  335.05  5449.5  338.68  5580.0  342.48  5685.0  343.52  5797.6  346.73
  5841.1  347.26  5881.2  349.18  5907.3  351.69  5931.4  351.34  5968.3  352.64
#Mann=6,-1,0
  4509.9    0.05       0  4901.4    0.12       0  4982.6    0.07       0
  4992.8    0.12       0  5263.9    0.05       0  5797.6    0.12       0
Bank Sta=4982.6,4992.8
Exp/Cntr=0.3,0.1

Type RM Length L Ch R = 1,11326,213,213,213
BEGIN DESCRIPTION:
Persimmon Branch 230
END DESCRIPTION:
XS GIS Cut Line= 3
      2676553.16      6817074.07      2676090.97      6817035.41
      2675205.13      6816907.00
#Sta/Elev= 30
  4544.5  347.75  4639.2  346.33  4712.2  343.05  4752.4  343.64  4842.7  338.90
  4903.5  336.59  4983.2  334.77  4993.2  333.30  5003.2  328.72  5004.6  328.22
  5012.0  328.22  5013.4  328.72  5023.4  331.78  5033.5  333.31  5063.8  333.14
  5084.1  331.95  5124.5  331.86  5134.6  332.53  5174.9  332.82  5326.6  334.56
  5417.4  336.04  5468.0  337.61  5548.9  338.42  5703.4  342.69  5740.9  345.00
  5768.5  345.27  5773.6  346.04  5831.8  346.62  5877.6  348.42  5903.4  349.47
#Mann=6,-1,0
  4544.5    0.05       0  4903.5    0.12       0  5003.2    0.07       0
  5013.4    0.12       0  5174.9    0.05       0  5877.6    0.12       0
Bank Sta=5003.2,5013.4
Exp/Cntr=0.3,0.1

Type RM Length L Ch R = 1,11113,219,219,219
BEGIN DESCRIPTION:
Persimmon Branch 231
END DESCRIPTION:
XS GIS Cut Line= 3
      2676572.45      6816999.16      2676178.85      6816847.71
      2675269.85      6816724.12
#Sta/Elev= 30
  4575.3  346.59  4689.4  343.84  4700.5  343.11  4774.4  340.88  4839.7  337.85
  4922.0  335.90  4949.0  335.89  4957.2  336.79  4973.6  334.40  4979.0  334.73
  4989.4  333.56  4995.9  328.09  5001.0  328.09  5007.2  327.28  5008.6  326.78
  5016.1  326.78  5017.5  327.28  5020.1  332.66  5040.3  332.83  5050.4  332.00
  5090.7  331.54  5149.5  332.07  5234.7  332.36  5625.6  338.16  5655.9  338.98
  5736.6  342.43  5777.0  344.74  5824.3  346.72  5896.7  348.65  5914.4  349.73
#Mann=5,-1,0
  4575.3    0.05       0  4922.0    0.12       0  5007.2    0.07       0
  5017.5    0.12       0  5149.5    0.05       0
Bank Sta=5007.2,5017.5
Exp/Cntr=0.3,0.1

Type RM Length L Ch R = 1,10894,292,292,292
BEGIN DESCRIPTION:
Persimmon Branch 229
END DESCRIPTION:
XS GIS Cut Line= 3
      2676620.06      6816937.83      2676266.68      6816662.60
      2675459.74      6816211.90
#Sta/Elev= 30
  4554.6  345.61  4711.9  341.92  4922.0  335.30  4990.7  334.32  4997.0  333.74
  4999.8  330.87  5005.8  330.87  5012.5  328.31  5018.3  327.89  5021.0  326.81
  5022.5  326.31  5030.0  326.31  5031.4  326.81  5049.1  332.94  5071.9  332.46
  5077.7  333.27  5106.4  331.43  5144.8  331.32  5239.9  332.61  5358.4  332.81
  5526.6  334.24  5591.7  335.55  5607.7  335.32  5716.2  337.73  5769.9  340.22
  5835.0  344.59  5885.3  346.58  5900.2  345.90  5916.1  347.21  5926.8  349.08
#Mann=5,-1,0
  4554.6    0.05       0  4922.0    0.12       0  5021.0    0.07       0
  5031.4    0.12       0  5144.8    0.05       0
Bank Sta=5021,5031.4
Exp/Cntr=0.3,0.1

Type RM Length L Ch R = 1,10602,300,300,300
BEGIN DESCRIPTION:
Persimmon Branch 33
END DESCRIPTION:
XS GIS Cut Line= 3
      2676775.98      6816511.00      2676376.00      6816411.00
      2675575.99      6816111.00
#Sta/Elev= 30
  4582.8  344.29  4613.7  343.44  4642.1  341.80  4770.9  338.17  4816.5  336.25
  4840.5  334.89  4953.9  333.14  4964.2  332.03  4971.9  328.43  4977.1  332.08
  4984.8  329.23  5011.2  325.75  5012.7  325.25  5021.7  325.75  5027.1  330.40
  5035.1  332.13  5090.3  331.15  5138.5  331.62  5358.2  332.87  5486.4  334.36
  5517.5  335.46  5553.1  335.06  5688.4  337.88  5742.7  339.61  5748.9  340.71
  5754.3  339.89  5828.1  344.00  5839.7  344.96  5846.8  349.06  5849.5  349.06
#Mann=5,-1,0
  4582.8    0.05       0  4816.5    0.12       0  5011.2    0.07       0
  5021.7    0.12       0  5138.5    0.05       0
Bank Sta=5011.2,5021.7
Exp/Cntr=0.3,0.1

Type RM Length L Ch R = 1,10302,318,318,318
BEGIN DESCRIPTION:
Persimmon Branch 183
END DESCRIPTION:
XS GIS Cut Line= 3
      2677069.32      6816446.36      2676539.64      6816195.80
      2675616.28      6815798.13
#Sta/Elev= 30
  4415.0  350.36  4617.8  345.95  4738.6  341.08  4761.3  340.51  4766.9  341.49
  4772.7  340.18  4797.6  338.56  4948.9  332.50  4954.4  331.38  4993.9  331.42
  5000.0  327.72  5005.7  327.43  5018.2  324.58  5019.7  324.08  5028.7  324.58
  5037.6  327.66  5052.5  330.77  5171.2  331.30  5351.1  332.21  5684.2  336.86
  5807.3  340.74  5865.3  343.79  5883.3  346.06  5906.9  345.11  5912.3  346.29
  5935.8  345.23  5941.3  347.06  5959.4  346.23  5964.8  347.91  6006.3  347.96
#Mann=5,-1,0
  4415.0    0.05       0  4797.6    0.12       0  5018.2    0.07       0
  5028.7    0.12       0  5171.2    0.05       0
Bank Sta=5018.2,5028.7
Exp/Cntr=0.3,0.1

Type RM Length L Ch R = 1,9984,266,266,266
BEGIN DESCRIPTION:
Persimmon Branch 182
END DESCRIPTION:
XS GIS Cut Line= 3
      2677208.73      6816387.02      2676701.22      6815932.64
      2675691.01      6815744.36
#Sta/Elev= 30
  4322.5  351.45  4463.0  348.65  4505.6  346.71  4548.3  345.72  4682.8  337.26
  4719.8  336.53  4774.8  334.31  4831.6  333.30  4909.4  330.45  4944.5  330.66
  4958.7  329.71  4980.4  331.41  4987.1  330.88  4994.6  327.06  5001.2  330.96
  5003.7  330.96  5009.0  326.25  5013.9  324.28  5015.3  323.78  5024.5  324.28
  5029.3  329.53  5037.2  330.20  5093.6  330.14  5532.0  333.73  5558.3  334.27
  5568.5  335.12  5660.0  335.38  5833.0  340.57  5995.7  348.88  6031.3  349.69
#Mann=5,-1,0
  4322.5    0.05       0  4719.8    0.12       0  5013.9    0.07       0
  5024.5    0.12       0  5093.6    0.05       0
Bank Sta=5013.9,5024.5
Exp/Cntr=0.3,0.1

Type RM Length L Ch R = 1,9718,457,457,457
BEGIN DESCRIPTION:
Persimmon Branch 151
END DESCRIPTION:
XS GIS Cut Line= 3
      2677607.50      6816304.86      2676872.68      6815755.42
      2676105.19      6814817.42
#Sta/Elev= 30
  4080.4  351.83  4191.9  351.48  4306.5  346.40  4442.0  344.70  4542.1  340.37
  4562.9  337.94  4577.5  339.32  4805.3  331.82  4877.6  329.58  4898.4  330.64
  4913.0  328.95  4977.6  329.54  4983.9  328.51  4991.8  323.18  4993.3  322.68
  5003.1  323.18  5013.2  323.73  5019.7  328.67  5041.9  329.85  5361.4  331.52
  5524.3  335.35  5538.7  336.31  5559.5  342.70  5723.9  341.98  5743.6  343.24
  5808.6  346.87  5880.3  346.12  5944.2  348.32  6142.3  358.68  6209.9  360.66
#Mann=5,-1,0
  4080.4    0.05       0  4805.3    0.12       0  4991.8    0.07       0
  5003.1    0.12       0  5743.6    0.05       0
Bank Sta=4991.8,5003.1
Exp/Cntr=0.3,0.1

Type RM Length L Ch R = 1,9261,939,939,939
BEGIN DESCRIPTION:
Persimmon Branch 150
END DESCRIPTION:
XS GIS Cut Line= 3
      2677773.43      6815975.98      2676979.40      6815446.04
      2676335.16      6814787.77
#Sta/Elev= 30
  4053.2  347.83  4069.7  348.69  4090.7  347.05  4126.7  347.36  4322.0  350.90
  4647.1  335.09  4682.5  332.94  4819.6  329.33  4832.7  328.17  4841.7  325.50
  4847.7  326.07  4855.6  329.11  4955.8  328.52  4991.9  329.44  5001.2  323.35
  5002.8  322.85  5012.5  323.35  5020.9  327.25  5028.0  328.38  5063.3  327.91
  5084.6  329.17  5176.5  328.23  5197.6  329.78  5254.2  329.54  5552.7  344.50
  5600.8  346.27  5621.9  345.92  5657.4  348.13  5720.9  348.25  5928.9  352.50
#Mann=5,-1,0
  4053.2    0.05       0  4647.1    0.12       0  5001.2    0.07       0
  5012.5    0.12       0  5552.7    0.05       0
Bank Sta=5001.2,5012.5
Exp/Cntr=0.3,0.1

Type RM Length L Ch R = 1,8322,145,145,145
BEGIN DESCRIPTION:
Persimmon Branch 149
END DESCRIPTION:
XS GIS Cut Line= 3
      2678261.47      6815169.27      2677479.95      6814875.12
      2676446.27      6814817.91
#Sta/Elev= 30
  4160.8  349.32  4348.3  343.81  4359.0  344.43  4380.3  342.50  4391.0  343.06
  4583.4  336.56  4710.8  330.60  4732.7  328.34  4775.7  326.93  4848.3  326.45
  4853.6  324.22  4871.8  324.45  4878.5  326.45  4914.6  325.61  4957.3  326.96
  4963.4  322.05  4965.0  321.55  4974.8  322.05  4988.7  326.53  5039.9  327.15
  5120.0  325.27  5190.1  327.24  5220.1  326.49  5323.1  328.04  5430.5  330.19
  5519.2  330.36  5600.7  333.95  5771.0  345.84  5841.1  348.89  6031.1  351.88
#Mann=5,-1,0
  4160.8    0.05       0  4710.8    0.12       0  4963.4    0.07       0
  4974.8    0.12       0  5323.1    0.05       0
Bank Sta=4963.4,4974.8
Exp/Cntr=0.3,0.1

Type RM Length L Ch R = 1,8177,461,461,461
BEGIN DESCRIPTION:
Persimmon Branch 148
END DESCRIPTION:
XS GIS Cut Line= 3
      2678375.19      6814811.58      2677518.09      6814744.34
      2676671.44      6814739.70
#Sta/Elev= 30
  4146.2  344.65  4245.7  344.09  4285.8  342.57  4305.9  340.29  4348.2  338.32
  4426.2  336.26  4446.3  337.10  4516.5  334.04  4556.6  333.89  4667.0  330.59
  4697.1  328.68  4753.7  328.35  4859.7  326.54  4937.8  326.90  4957.9  325.50
  5009.5  326.16  5022.3  321.78  5023.9  321.28  5033.7  321.78  5058.0  321.93
  5078.0  326.25  5128.0  323.26  5138.0  325.05  5168.0  326.52  5278.5  327.52
  5348.0  327.78  5508.0  331.79  5588.0  332.48  5648.0  334.65  5852.6  346.60
#Mann=5,-1,0
  4146.2    0.05       0  4753.7    0.12       0  5022.3    0.07       0
  5033.7    0.12       0  5278.5    0.05       0
Bank Sta=5022.3,5033.7
Exp/Cntr=0.3,0.1

Type RM Length L Ch R = 1,7716,471,471,471
BEGIN DESCRIPTION:
Persimmon Branch 152
END DESCRIPTION:
XS GIS Cut Line= 3
      2678527.88      6814566.41      2677582.29      6814447.02
      2677284.86      6813526.16
#Sta/Elev= 30
  4292.2  341.87  4435.2  336.57  4576.3  333.93  4657.0  334.60  4833.9  329.10
  4969.4  325.53  4979.5  324.87  4994.0  321.72  4995.5  321.22  5005.4  321.72
  5014.4  321.76  5029.9  324.82  5188.8  325.50  5253.2  324.68  5451.3  326.88
  5541.5  326.58  5756.0  332.18  5936.3  342.23  5963.1  337.61  5995.1  342.66
  6000.4  341.22  6027.2  345.59  6032.4  344.63  6050.3  347.71  6064.5  347.64
  6113.3  354.03  6155.3  358.04  6160.6  357.45  6192.6  362.30  6213.0  362.75
#Mann=5,-1,0
  4292.2    0.05       0  4833.9    0.12       0  4994.0    0.07       0
  5005.4    0.12       0  5188.8    0.05       0
Bank Sta=4994,5005.4
Exp/Cntr=0.3,0.1

Type RM Length L Ch R = 1,7245,715,715,715
BEGIN DESCRIPTION:
Persimmon Branch 147
END DESCRIPTION:
XS GIS Cut Line= 3
      2678703.00      6814610.94      2677780.09      6814057.38
      2677220.71      6813297.46
#Sta/Elev= 30
  3923.6  346.87  4374.7  334.40  4380.5  332.90  4503.1  328.59  4635.2  328.13
  4678.1  326.40  4687.7  322.37  4693.7  322.00  4703.2  321.98  4704.8  321.48
  4714.8  321.98  4730.4  322.04  4746.0  324.93  4948.1  323.87  4969.6  322.00
  4992.9  322.02  4999.3  323.74  5032.3  323.17  5100.2  323.62  5114.8  322.00
  5135.7  324.72  5206.6  326.10  5392.6  337.99  5479.6  341.12  5687.2  368.63
  5737.3  373.88  5772.8  374.16  5843.8  369.09  5893.9  368.83  5943.4  371.33
#Mann=5,-1,0
  3923.6    0.05       0  4693.7    0.12       0  4703.2    0.07       0
  4714.8    0.12       0  5032.3    0.05       0
Bank Sta=4703.2,4714.8
Exp/Cntr=0.3,0.1

Type RM Length L Ch R = 1,6530,930,930,930
BEGIN DESCRIPTION:
Persimmon Branch 146
END DESCRIPTION:
XS GIS Cut Line= 3
      2678868.95      6814552.25      2678293.47      6813708.41
      2677326.08      6813085.28
#Sta/Elev= 30
  4004.6  345.09  4195.0  336.76  4287.7  337.86  4404.3  335.67  4503.2  330.30
  4670.6  326.78  4676.6  326.47  4683.9  322.15  4698.4  322.00  4784.4  322.13
  4805.3  324.22  4850.1  322.34  5226.6  321.87  5228.2  321.37  5238.2  321.87
  5247.7  322.15  5450.2  325.25  5471.3  327.36  5522.6  327.90  5607.3  332.02
  5674.0  339.50  5737.4  348.69  5861.5  362.24  5934.1  371.65  5970.4  372.26
  5994.6  370.82  6027.9  369.12  6106.4  368.92  6172.1  373.62  6176.7  373.51
#Mann=7,-1,0
  4004.6    0.05       0  4698.4     0.1       0  5226.6    0.07       0
  5238.2     0.1       0  5247.7    0.05       0  5994.6    0.12       0
  6172.1    0.05       0
Bank Sta=5226.6,5238.2
Exp/Cntr=0.3,0.1

Type RM Length L Ch R = 1,5600,792,792,792
BEGIN DESCRIPTION:
Persimmon Branch 145
END DESCRIPTION:
XS GIS Cut Line= 3
      2679395.89      6814120.45      2678869.88      6813166.88
      2677951.72      6812185.29
#Sta/Elev= 30
  3910.2  341.27  3967.1  342.28  4042.7  340.42  4129.8  341.55  4395.7  337.89
  4549.1  330.24  4586.0  326.03  4602.0  326.38  4613.4  325.07  4639.9  324.33
  4661.5  322.00  4663.1  321.50  4673.2  322.00  5416.7  322.00  5425.0  322.92
  5508.5  324.41  5678.2  334.38  5862.2  357.90  5925.7  363.26  5968.2  364.89
  6010.7  364.33  6102.7  359.26  6124.0  359.69  6145.0  358.08  6152.3  359.54
  6159.2  358.36  6187.5  358.73  6251.5  361.46  6286.7  361.37  6343.3  364.85
#Mann=5,-1,0
  3910.2    0.05       0  4613.4     0.1       0  4661.5    0.07       0
  4673.2     0.1       0  5425.0    0.05       0
Bank Sta=4661.5,4673.2
Exp/Cntr=0.3,0.1

Type RM Length L Ch R = 1,4808,509,509,509
BEGIN DESCRIPTION:
Persimmon Branch 144
END DESCRIPTION:
XS GIS Cut Line= 3
      2679631.05      6813855.47      2679463.18      6812660.36
      2678265.73      6811775.59
#Sta/Elev= 30
  3790.0  338.35  3915.7  336.51  3946.0  333.91  4188.3  328.54  4299.4  328.56
  4596.5  322.00  4598.1  321.50  4608.2  322.00  5517.3  322.00  5549.5  322.00
  5580.1  322.00  5588.5  323.69  5594.8  323.34  5602.6  327.99  5624.0  329.51
  5724.2  330.24  5730.4  328.43  5751.8  327.99  5824.4  329.22  5880.8  331.93
  5945.5  332.20  5950.4  333.46  5988.0  335.27  5995.6  334.35  6021.8  335.16
  6166.8  342.52  6196.1  342.82  6346.4  350.79  6373.5  353.58  6485.7  358.80
#Mann=7,-1,0
  3790.0    0.05       0  4596.5    0.03       0  4608.2    0.05       0
  5517.3     0.1       0  5549.5    0.05       0  5950.4   0.075       0
  6021.8    0.05       0
Bank Sta=4596.5,4608.2
Exp/Cntr=0.3,0.1

Type RM Length L Ch R = 1,4299,509,509,509
BEGIN DESCRIPTION:
Persimmon Branch 128
END DESCRIPTION:
XS GIS Cut Line= 3
      2679808.97      6814001.10      2679908.88      6812462.07
      2679698.69      6810985.73
#Sta/Elev= 30
  3457.8  343.48  3688.4  338.91  3738.5  338.80  3808.6  341.06  3858.7  340.24
  3953.1  336.19  4029.1  330.54  4209.5  323.18  4213.4  322.00  4215.1  321.50
  4225.7  322.00  5769.7  322.00  5790.8  323.18  5829.4  324.46  5835.4  326.62
  5840.5  325.08  5849.6  325.30  5910.5  329.78  5977.1  337.53  6001.1  337.82
  6011.2  340.02  6038.7  342.49  6152.6  354.42  6189.6  355.77  6194.6  357.05
  6233.5  356.84  6294.1  358.91  6336.5  361.81  6431.8  369.87  6491.3  372.68
#Mann=8,-1,0
  3457.8    0.05       0  4213.4    0.03       0  4225.7    0.05       0
  5790.8     0.1       0  5910.5   0.075       0  6038.7    0.05       0
  6336.5   0.075       0  6431.8    0.05       0
Bank Sta=4213.4,4225.7
Exp/Cntr=0.3,0.1

Type RM Length L Ch R = 1,3790,752,752,752
BEGIN DESCRIPTION:
Persimmon Branch 129
END DESCRIPTION:
XS GIS Cut Line= 3
      2680068.91      6814214.67      2680402.50      6812412.29
      2679716.06      6810526.96
#Sta/Elev= 30
  3164.9  348.49  3291.0  346.78  3338.8  344.56  3361.9  346.27  3391.7  345.96
  3425.4  344.03  3443.2  344.86  3454.8  342.89  3544.9  342.92  3692.6  334.49
  3809.3  328.71  3972.1  324.32  3986.2  322.00  3987.9  321.50  3998.5  322.00
  5964.6  322.00  5989.0  324.79  6112.2  331.82  6234.5  343.67  6286.8  346.68
  6439.9  355.07  6499.8  359.60  6519.0  359.36  6549.6  361.79  6554.9  363.54
  6601.0  365.22  6662.7  367.98  6758.3  370.16  6925.5  367.36  7004.3  369.60
#Mann=9,-1,0
  3164.9    0.05       0  3425.4    0.12       0  3692.6    0.05       0
  3986.2    0.03       0  3998.5    0.05       0  6286.8   0.075       0
  6439.9    0.05       0  6601.0   0.075       0  6662.7    0.05       0
Bank Sta=3986.2,3998.5
Exp/Cntr=0.3,0.1

Type RM Length L Ch R = 1,3038,951,951,951
BEGIN DESCRIPTION:
Persimmon Branch 102
END DESCRIPTION:
XS GIS Cut Line= 3
      2681151.17      6814731.60      2681138.99      6812341.54
      2680016.26      6810439.70
#Sta/Elev= 30
  2629.4  343.45  2670.0  343.02  2810.0  334.58  2850.0  333.73  2910.0  330.15
  3010.0  326.31  3020.0  322.18  3023.8  322.00  3025.5  321.50  3036.3  322.00
  6532.9  322.00  6541.4  325.66  6554.3  327.05  6649.9  332.75  6724.1  336.15
  6751.4  338.57  6782.7  339.38  6809.9  341.97  6905.5  347.54  6994.2  350.30
  7022.6  352.58  7038.3  352.54  7044.1  353.62  7059.7  353.20  7081.2  354.16
  7096.8  353.39  7102.6  354.24  7145.5  354.92  7198.2  354.50  7228.0  355.36
#Mann=3,-1,0
  2629.4    0.05       0  3023.8    0.03       0  3036.3    0.05       0
Bank Sta=3023.8,3036.3
Exp/Cntr=0.3,0.1

Type RM Length L Ch R = 1,2087,606,606,606
BEGIN DESCRIPTION:
Persimmon Branch 91
END DESCRIPTION:
XS GIS Cut Line= 3
      2681484.52      6815481.91      2682081.86      6812386.56
      2680036.90      6810099.02
#Sta/Elev= 30
  1813.2  345.82  1854.9  344.15  1895.3  344.22  1936.3  342.89  1957.4  341.18
  2107.8  337.26  2150.2  334.41  2191.0  334.26  2216.6  331.80  2221.7  332.28
  2252.1  328.37  2262.2  322.00  2264.0  321.50  2274.8  322.00  7261.4  322.00
  7275.6  324.02  7367.5  327.99  7445.3  332.90  7579.9  338.78  7757.1  341.50
  7778.0  343.49  7792.2  344.12  7799.7  343.40  7834.8  345.57  7905.9  346.31
  7912.6  347.38  7941.0  348.11  7962.7  347.77  7983.6  349.97  8034.0  351.92
#Mann=3,-1,0
  1813.2    0.05       0  2262.2    0.03       0  2274.8    0.05       0
Bank Sta=2262.2,2274.8
Exp/Cntr=0.3,0.1

Type RM Length L Ch R = 1,1481,469,469,469
BEGIN DESCRIPTION:
Persimmon Branch 32
END DESCRIPTION:
XS GIS Cut Line= 5
      2681410.51      6816172.96      2683110.11      6814764.34
      2682930.86      6812890.13      2682626.00      6812261.00
      2680226.02      6809861.02
#Sta/Elev= 30
   211.1  348.08   252.0  345.36   301.5  345.37   315.8  343.91   351.0  344.31
   394.0  342.91   457.8  343.40   472.1  342.04   507.3  342.18   628.4  337.31
   749.5  334.51   877.2  329.29   933.1  327.98   969.6  323.62   976.1  323.65
   977.4  322.00   979.3  321.50   990.5  322.00  7729.8  322.00  7843.0  328.90
  7871.3  328.87  7913.7  331.05  7927.8  330.47  8097.5  337.88  8140.0  337.84
  8168.3  339.81  8281.4  341.88  8309.7  344.69  8323.8  344.38  8394.5  349.23
#Mann=3,-1,0
   211.1    0.05       0   977.4    0.03       0   990.5    0.05       0
Bank Sta=977.4,990.5
Exp/Cntr=0.3,0.1

Type RM Length L Ch R = 1,1012,495,495,495
BEGIN DESCRIPTION:
Persimmon Branch 31
END DESCRIPTION:
XS GIS Cut Line= 4
      2681436.69      6816320.71      2683331.11      6814899.86
      2682976.00      6811961.00      2680576.00      6809561.00
#Sta/Elev= 30
  -328.0  343.38  -228.9  341.82  -221.4  340.72  -215.1  341.25  -192.2  339.79
  -100.5  338.04   -78.9  336.19    71.1  335.26   114.0  333.63   128.6  331.80
   149.5  332.18   278.6  325.70   314.0  325.65   328.6  324.00   334.9  324.88
   336.7  322.00   338.5  321.50   349.8  322.00  7814.6  322.00  7828.7  323.95
  7842.9  323.79  7871.1  327.30  7899.4  328.09  7927.7  330.90  8040.8  333.62
  8069.1  335.99  8182.3  336.02  8238.8  337.35  8366.1  344.26  8394.4  344.61
#Mann=3,-1,0
  -328.0    0.05       0   336.7    0.03       0   349.8    0.05       0
Bank Sta=336.7,349.8
Exp/Cntr=0.3,0.1

Type RM Length L Ch R = 1,517,0,0,0
BEGIN DESCRIPTION:
Persimmon Branch 30
END DESCRIPTION:
XS GIS Cut Line= 4
      2681374.67      6816466.55      2683640.25      6815390.79
      2683326.00      6811611.00      2680326.02      6808911.02
#Sta/Elev= 30
 -1300.5  344.19 -1160.0  339.81 -1040.8  339.32  -876.2  326.52  -859.0  322.00
  -853.5  324.19  -845.2  322.00  -807.4  321.89  -805.6  321.39  -794.3  321.89
  -762.6  323.55  -745.5  322.00  7581.5  322.00  7770.2  322.00  7893.0  322.00
  7946.3  322.00  7953.0  323.90  7967.2  322.38  7974.0  325.82  7981.4  325.76
  7995.1  329.21  8052.4  330.55  8149.2  329.28  8285.6  329.33  8314.0  332.03
  8391.8  334.97  8441.9  338.52  8625.7  346.31  8668.3  349.89  9036.4  367.14
#Mann=8,-1,0
 -1300.5    0.05       0  -807.4    0.03       0  -794.3    0.05       0
  7581.5     0.1       0  7770.2   0.075       0  7893.0     0.1       0
  7995.1   0.075       0  8149.2    0.05       0
Bank Sta=-807.4,-794.3
Exp/Cntr=0.3,0.1

Chan Stop Cuts=-1
