--- Prairie Creek.prj (project) ---

Proj Title=Prairie Creek Base Level Engineering
Current Plan=p01
Default Exp/Contr=0.3,0.1
English Units
Geom File=g01
Flow File=f01
Plan File=p01
BEGIN DESCRIPTION:
Prairie Creek
END DESCRIPTION:

--- Prairie Creek.p01 (plan) ---

Plan Title=Multiple Run
Short Identifier=Multiple
Geom File=g01
Flow File=f01
Subcritical Flow
K Sum by GR= 0
Std Step Tol= 0.01
Critical Tol= 0.01
Num of Std Step Trials= 20
Max Error Tol= 0.3
Flow Tol Ratio= 0.001
Split Flow NTrial= 30
Split Flow Tol= 0.02
Split Flow Ratio= 0.02
Log Output Level= 0
Friction Slope Method= 1
Unsteady Friction Slope Method= 2
Unsteady Bridges Friction Slope Method= 1
Parabolic Critical Depth
Global Vel Dist=  1 , 1 , 1
Global Log Level= 0
CheckData=True
Encroach Param= -1, 0, 0, 0
BEGIN DESCRIPTION:
Multiple Run
END DESCRIPTION:

--- Prairie Creek.f01 (steady flow) ---

Flow Title=Multiple
Number of Profiles=7
Profile Names=10-year,25-year,50-year,1pct_min,100-year,1pct_plu,500-year
River Rch & RM= Prairie Creek,Reach-1,63568
     651     874    1055     631    1259    2513    1793
River Rch & RM= Prairie Creek,Reach-1,60487
     780    1056    1281     769    1535    3063    2206
River Rch & RM= Prairie Creek,Reach-1,59050
     958    1303    1585     954    1904    3799    2748
River Rch & RM= Prairie Creek,Reach-1,55454
    1072    1454    1763    1057    2109    4209    3020
River Rch & RM= Prairie Creek,Reach-1,47344
    1452    2000    2453    1485    2962    5911    4325
River Rch & RM= Prairie Creek,Reach-1,45731
    1593    2203    2708    1643    3278    6541    4809
River Rch & RM= Prairie Creek,Reach-1,42817
    1756    2435    2998    1821    3634    7250    5343
River Rch & RM= Prairie Creek,Reach-1,40719
    1796    2485    3055    1852    3696    7375    5415
River Rch & RM= Prairie Creek,Reach-1,31958
    2309    3224    3989    2432    4852    9682    7188
River Rch & RM= Prairie Creek,Reach-1,22159
    2447    3424    4241    2588    5164   10304    7665
River Rch & RM= Prairie Creek,Reach-1,21201
    2453    3428    4243    2587    5162   10300    7649
River Rch & RM= Prairie Creek,Reach-1,18495
    2682    3761    4666    2851    5689   11351    8466
River Rch & RM= Prairie Creek,Reach-1,17956
    2668    3737    4632    2828    5643   11259    8382
River Rch & RM= Prairie Creek,Reach-1,16082
    2800    3929    4877    2981    5948   11868    8856
River Rch & RM= Prairie Creek,Reach-1,15448
    2843    3986    4945    3021    6027   12026    8962
River Rch & RM= Prairie Creek,Reach-1,12827
    2863    4014    4979    3041    6068   12108    9021
River Rch & RM= Prairie Creek,Reach-1,11691
    2890    4051    5023    3067    6119   12210    9090
River Rch & RM= Prairie Creek,Reach-1,10111
    2880    4033    4998    3050    6086   12143    9031
River Rch & RM= Prairie Creek,Reach-1,9082
    3018    4230    5246    3203    6391   12752    9492
River Rch & RM= Prairie Creek,Reach-1,7755
    3020    4228    5237    3194    6373   12716    9445
River Rch & RM= Prairie Creek,Reach-1,5045
    2989    4170    5154    3136    6257   12485    9228
Boundary for River Rch & Prof#=Prairie Creek,Reach-1,1
Up Type=0
Dn Type=3
Dn Slope=0.005
Boundary for River Rch & Prof#=Prairie Creek,Reach-1,2
Up Type=0
Dn Type=3
Dn Slope=0.005
Boundary for River Rch & Prof#=Prairie Creek,Reach-1,3
Up Type=0
Dn Type=3
Dn Slope=0.005
Boundary for River Rch & Prof#=Prairie Creek,Reach-1,4
Up Type=0
Dn Type=3
Dn Slope=0.005
Boundary for River Rch & Prof#=Prairie Creek,Reach-1,5
Up Type=0
Dn Type=3
Dn Slope=0.005
Boundary for River Rch & Prof#=Prairie Creek,Reach-1,6
Up Type=0
Dn Type=3
Dn Slope=0.005
Boundary for River Rch & Prof#=Prairie Creek,Reach-1,7
Up Type=0
Dn Type=3
Dn Slope=0.005

--- Prairie Creek.g01 (geometry) ---

Geom Title=Existing Conditions

River Reach=Prairie Creek,Reach-1
Reach XY= 30
      2717176.00      6836211.00      2715881.26      6836808.91
      2711832.75      6834320.10      2710873.53      6834405.55
      2709089.76      6832724.24      2708586.94      6832721.44
      2708825.02      6832071.27      2708223.91      6830216.26
      2707442.71      6829227.56      2706016.35      6828612.36
      2703877.98      6828607.96      2702681.52      6827163.44
      2701922.63      6824512.22      2701125.71      6823583.77
      2701672.86      6823159.36      2701581.04      6822515.93
      2702672.73      6822009.64      2703068.51      6821011.03
      2702676.55      6819921.63      2703118.51      6819557.38
      2702022.77      6817419.01      2701143.15      6816627.28
      2699386.63      6816221.12      2699070.94      6814608.75
      2697185.15      6812017.73      2697124.62      6807870.66
      2695927.36      6804651.35      2695722.46      6801462.46
      2694228.06      6799905.15      2694176.00      6797461.00

Type RM Length L Ch R = 1,63568,301,301,301
BEGIN DESCRIPTION:
Prairie Creek63568.221
END DESCRIPTION:
XS GIS Cut Line= 3
      2716939.12      6835774.91      2717132.15      6836213.29
      2717381.03      6836882.51
#Sta/Elev= 30
  4521.0  418.77  4576.1  418.95  4622.7  414.25  4651.5  414.55  4658.8  413.28
  4680.6  412.51  4866.4  410.33  4900.1  410.82  4971.3  409.19  4986.6  410.42
  4994.6  406.41  4998.6  406.17  5008.2  408.26  5040.2  409.07  5047.8  405.21
  5048.1  404.71  5051.8  405.21  5061.6  408.38  5080.2  409.37  5218.9  410.11
  5232.3  410.01  5256.9  411.80  5296.3  410.83  5353.2  411.74  5453.4  412.77
  5477.7  414.20  5508.7  413.33  5605.7  413.66  5691.1  414.41  5714.0  415.52
#Mann=6,-1,0
  4521.0    0.05       0  4900.1    0.12       0  5047.8    0.07       0
  5051.8    0.12       0  5218.9    0.16       0  5353.2    0.05       0
Bank Sta=5047.8,5051.8
Exp/Cntr=0.3,0.1

Type RM Length L Ch R = 1,63267,332,332,332
BEGIN DESCRIPTION:
Prairie Creek63267
END DESCRIPTION:
XS GIS Cut Line= 3
      2716755.12      6836044.14      2716876.52      6836258.20
      2717113.21      6836824.75
#Sta/Elev= 30
  4752.7  412.32  4798.3  411.59  4921.3  409.98  4927.0  409.81  4933.0  408.72
  4948.1  410.02  4962.1  409.63  4979.0  407.93  5008.8  406.59  5012.2  405.57
  5012.5  405.07  5016.0  405.07  5016.2  405.57  5032.6  407.77  5058.3  407.00
  5061.9  406.73  5085.7  410.99  5109.5  406.45  5121.0  405.78  5165.5  405.96
  5186.1  408.08  5268.6  408.03  5283.6  408.78  5316.1  409.05  5327.0  410.20
  5350.9  409.30  5369.2  409.85  5467.8  410.32  5557.6  412.52  5612.8  411.89
#Mann=8,-1,0
  4752.7    0.05       0  4798.3    0.07       0  4948.1    0.16       0
  4962.1    0.12       0  5012.2    0.07       0  5016.2    0.12       0
  5058.3    0.16       0  5165.5    0.05       0
Bank Sta=5012.2,5016.2
Exp/Cntr=0.3,0.1

Type RM Length L Ch R = 1,62935,439,439,439
BEGIN DESCRIPTION:
Prairie Creek62934.95
END DESCRIPTION:
XS GIS Cut Line= 3
      2716517.68      6836146.02      2716656.86      6836481.72
      2716886.64      6837093.17
#Sta/Elev= 30
  4638.5  411.45  4648.2  411.70  4654.7  410.93  4677.5  409.93  4773.1  410.04
  4778.5  409.11  4802.3  409.40  4849.6  408.36  4884.8  408.48  4932.6  407.72
  4968.6  408.41  4995.7  407.04  5086.6  406.39  5130.6  406.72  5138.0  406.16
  5138.3  405.66  5141.8  405.66  5142.0  406.16  5216.4  407.02  5257.5  408.96
  5271.5  407.74  5289.6  407.69  5301.8  408.33  5343.0  408.20  5361.9  408.73
  5370.5  408.74  5522.3  409.68  5552.5  410.84  5588.7  410.15  5655.1  410.40
#Mann=7,-1,0
  4638.5    0.07       0  4995.7    0.12       0  5130.6    0.05       0
  5138.0    0.07       0  5142.0    0.05       0  5361.9    0.12       0
  5370.5    0.05       0
Bank Sta=5138,5142
Exp/Cntr=0.3,0.1

Type RM Length L Ch R = 1,62496,148,148,148
BEGIN DESCRIPTION:
Prairie Creek62495.75
END DESCRIPTION:
XS GIS Cut Line= 4
      2716403.38      6836132.96      2716385.91      6836762.94
      2716420.88      6837189.69      2716513.02      6837516.66
#Sta/Elev= 30
  4371.6  411.02  4456.0  409.83  4487.2  410.10  4519.7  409.57  4529.7  408.65
  4559.7  408.05  4619.7  408.15  4833.5  406.58  4879.8  405.90  4931.4  405.91
  4939.9  405.54  4959.9  406.61  4979.9  406.08  5001.8  406.30  5009.9  404.18
  5017.9  403.04  5018.2  402.54  5021.7  402.54  5021.9  403.04  5030.0  404.84
  5040.0  404.51  5059.6  406.63  5064.6  406.04  5195.2  407.11  5462.3  408.61
  5493.7  409.04  5506.7  410.07  5540.7  409.40  5545.9  408.86  5769.7  409.75
#Mann=7,-1,0
  4371.6    0.07       0  4487.2    0.05       0  4833.5    0.16       0
  4931.4    0.12       0  5017.9    0.07       0  5021.9    0.12       0
  5195.2    0.05       0
Bank Sta=5017.9,5021.9
Exp/Cntr=0.3,0.1

Type RM Length L Ch R = 1,62348,364,364,364
BEGIN DESCRIPTION:
Prairie Creek62348.46
END DESCRIPTION:
XS GIS Cut Line= 4
      2716231.92      6836177.52      2716238.82      6836769.94
      2716221.91      6837154.13      2716012.95      6837551.06
#Sta/Elev= 30
  4415.6  409.41  4489.1  409.19  4529.1  408.04  4599.1  407.58  4879.1  406.52
  4927.1  405.17  4949.1  404.63  4967.1  402.66  4967.4  402.16  4970.9  402.16
  4971.1  402.66  4979.1  404.54  5025.1  404.99  5159.3  404.04  5169.3  404.09
  5185.1  406.40  5222.7  405.84  5392.6  407.24  5438.7  405.30  5490.8  404.42
  5536.0  404.29  5548.9  405.26  5570.9  404.75  5603.7  405.29  5615.1  404.19
  5647.8  405.95  5653.4  407.25  5659.9  407.49  5770.5  408.11  5841.2  408.33
#Mann=8,-1,0
  4415.6    0.05       0  4927.1    0.16       0  4967.1    0.07       0
  4971.1    0.16       0  5025.1    0.12       0  5222.7    0.05       0
  5659.9    0.07       0  5770.5    0.05       0
Bank Sta=4967.1,4971.1
Exp/Cntr=0.3,0.1

Type RM Length L Ch R = 1,61984,436,436,436
BEGIN DESCRIPTION:
Prairie Creek61983.9
END DESCRIPTION:
XS GIS Cut Line= 3
      2716082.92      6836060.62      2715889.22      6836814.70
      2715770.79      6837372.00
#Sta/Elev= 30
  4225.7  409.70  4267.4  409.94  4288.0  408.69  4401.6  407.39  4517.6  406.96
  4535.8  407.84  4558.3  406.65  4716.1  405.01  4732.0  405.72  4773.3  404.29
  4845.6  404.93  4866.7  404.61  4879.1  404.25  4897.2  402.79  4919.9  402.18
  4967.2  402.26  4996.2  402.99  5000.7  400.79  5008.7  400.78  5008.9  400.28
  5012.4  400.28  5012.7  400.78  5020.9  402.11  5040.0  402.41  5045.1  403.75
  5139.3  405.40  5183.8  406.13  5520.8  407.34  5552.5  407.77  5574.0  410.14
#Mann=5,-1,0
  4225.7    0.05       0  4866.7    0.12       0  4967.2    0.05       0
  5008.7    0.05       0  5012.7    0.05       0
Bank Sta=5008.7,5012.7
Exp/Cntr=0.3,0.1

Type RM Length L Ch R = 1,61548,612,612,612
BEGIN DESCRIPTION:
Prairie Creek61548.34
END DESCRIPTION:
XS GIS Cut Line= 3
      2715841.00      6835847.26      2715559.09      6836604.47
      2715318.40      6837295.05
#Sta/Elev= 30
  4199.7  410.98  4214.4  409.60  4259.7  408.24  4321.1  408.87  4345.4  407.22
  4417.1  406.36  4523.8  406.22  4555.8  407.23  4572.1  406.97  4577.4  406.08
  4651.9  405.75  4682.7  404.48  4859.4  403.13  4897.3  401.42  4939.7  400.97
  4952.0  401.74  4993.3  401.52  5000.4  402.78  5007.7  402.89  5012.6  400.02
  5012.8  399.52  5016.6  400.02  5032.7  400.93  5062.4  402.97  5093.5  402.65
  5217.8  404.50  5480.6  404.84  5580.2  405.40  5606.0  406.35  5739.0  406.35
#Mann=5,-1,0
  4199.7    0.05       0  4952.0    0.12       0  5012.6    0.07       0
  5016.6    0.12       0  5032.7    0.05       0
Bank Sta=5012.6,5016.6
Exp/Cntr=0.3,0.1

Type RM Length L Ch R = 1,60936,449,449,449
BEGIN DESCRIPTION:
Prairie Creek60935.94
END DESCRIPTION:
XS GIS Cut Line= 3
      2715232.49      6835474.77      2715161.21      6836273.20
      2715080.26      6837300.01
#Sta/Elev= 30
  4210.7  406.56  4317.3  406.03  4347.5  406.47  4417.7  405.63  4588.4  404.92
  4680.6  405.10  4787.0  404.10  4839.4  404.43  4859.5  403.83  4889.6  404.12
  4898.4  403.53  4949.9  402.66  4969.9  400.08  5000.1  399.28  5006.7  396.62
  5006.9  396.12  5010.4  396.12  5010.7  396.62  5020.1  398.66  5030.2  400.07
  5040.2  400.18  5070.3  401.95  5143.9  401.39  5250.8  402.29  5381.2  402.19
  5551.8  404.38  5742.4  404.95  5852.7  404.39  5872.8  404.90  6042.3  405.29
#Mann=3,-1,0
  4210.7    0.05       0  5006.7    0.05       0  5010.7    0.05       0
Bank Sta=5006.7,5010.7
Exp/Cntr=0.3,0.1

Type RM Length L Ch R = 1,60487,394,394,394
BEGIN DESCRIPTION:
Prairie Creek60486.73
END DESCRIPTION:
XS GIS Cut Line= 3
      2714774.80      6835443.44      2714711.39      6836283.62
      2714635.93      6837267.46
#Sta/Elev= 30
  4180.1  404.22  4879.6  402.03  4939.8  400.45  4959.9  398.53  5000.0  396.79
  5007.9  395.26  5008.2  394.76  5012.1  395.26  5018.8  397.74  5022.8  397.76
  5031.4  399.93  5089.8  399.52  5130.4  400.49  5162.0  399.92  5170.5  400.66
  5200.6  400.40  5230.7  401.54  5270.8  399.34  5287.5  399.84  5292.5  401.13
  5361.0  400.76  5371.1  401.58  5441.3  402.51  5702.0  403.21  5722.1  404.14
  5742.2  403.35  5922.7  404.29  5945.4  405.34  5962.8  404.31  6009.4  404.92
#Mann=5,-1,0
  4180.1    0.05       0  5007.9    0.05       0  5012.1    0.05       0
  5022.8    0.12       0  5089.8    0.05       0
Bank Sta=5007.9,5012.1
Exp/Cntr=0.3,0.1

Type RM Length L Ch R = 1,60093,545,545,545
BEGIN DESCRIPTION:
Prairie Creek60092.82
END DESCRIPTION:
XS GIS Cut Line= 3
      2714509.66      6835281.47      2714360.51      6836208.01
      2714230.41      6837264.87
#Sta/Elev= 30
  4073.0  404.28  4366.3  402.56  4447.3  400.50  4548.6  399.44  4619.5  400.07
  4771.4  399.39  4818.3  400.29  4823.4  399.49  4903.7  399.34  4942.0  400.00
  4974.0  397.25  4992.1  394.12  4992.4  393.62  4996.4  394.12  5003.8  397.53
  5008.9  396.13  5011.5  397.19  5056.2  399.94  5074.9  400.06  5084.6  399.13
  5175.9  400.74  5296.6  400.53  5387.3  401.65  5639.2  402.14  5663.3  402.99
  5689.5  402.41  5881.0  403.29  5901.1  404.35  5931.3  403.70  6076.3  404.43
#Mann=5,-1,0
  4073.0    0.05       0  4903.7    0.12       0  4992.1    0.07       0
  4996.4    0.12       0  5056.2    0.05       0
Bank Sta=4992.1,4996.4
Exp/Cntr=0.3,0.1

Type RM Length L Ch R = 1,59548,498,498,498
BEGIN DESCRIPTION:
Prairie Creek59548.45
END DESCRIPTION:
XS GIS Cut Line= 3
      2714105.73      6835098.83      2714074.72      6835808.13
      2714032.92      6836987.51
#Sta/Elev= 30
  4292.5  402.95  4444.8  402.73  4585.0  402.03  4665.0  400.81  4725.1  400.88
  4845.2  398.50  4895.2  398.16  4935.3  397.07  4955.3  395.76  4973.1  396.90
  4985.3  396.87  4993.0  393.57  4993.3  393.07  4997.3  393.07  4997.7  393.57
  5001.4  395.56  5006.4  395.56  5015.4  396.63  5055.4  396.51  5093.1  398.50
  5115.4  399.04  5275.5  398.98  5425.6  400.15  5475.6  399.28  5625.7  399.70
  5765.8  401.01  5925.9  401.51  5952.7  400.99  6096.0  402.22  6182.6  402.15
#Mann=5,-1,0
  4292.5    0.05       0  4973.1    0.12       0  4993.0    0.07       0
  4997.7    0.12       0  5093.1    0.05       0
Bank Sta=4993,4997.7
Exp/Cntr=0.3,0.1

Type RM Length L Ch R = 1,59050,331,331,331
BEGIN DESCRIPTION:
Prairie Creek59050.07
END DESCRIPTION:
XS GIS Cut Line= 3
      2713673.90      6835188.45      2713672.59      6835565.09
      2713677.96      6836927.53
#Sta/Elev= 30
  4628.1  405.59  4700.7  403.06  4820.7  401.52  4980.7  398.02  4990.7  396.58
  5000.2  394.15  5004.8  394.15  5008.1  392.12  5008.5  391.62  5013.3  392.12
  5050.7  395.92  5080.7  394.99  5150.7  396.84  5200.7  396.80  5270.7  399.46
  5298.7  398.02  5370.7  397.66  5390.7  398.93  5400.7  398.73  5410.7  397.46
  5467.6  398.01  5520.7  400.12  5570.7  399.58  5590.7  397.86  5750.7  399.47
  5850.7  399.32  5980.7  401.17  6030.7  400.33  6240.7  401.76  6367.2  401.73
#Mann=5,-1,0
  4628.1    0.05       0  5008.1    0.05       0  5013.3    0.05       0
  5298.7    0.16       0  5467.6    0.05       0
Bank Sta=5008.1,5013.3
Exp/Cntr=0.3,0.1

Type RM Length L Ch R = 1,58719,269,269,269
BEGIN DESCRIPTION:
Prairie Creek58719.31
END DESCRIPTION:
XS GIS Cut Line= 3
      2713465.34      6835153.32      2713382.86      6835545.45
      2713155.78      6836795.79
#Sta/Elev= 30
  4622.2  403.19  4838.6  400.78  4865.1  401.03  4883.3  399.79  4938.3  398.30
  4967.3  395.49  4983.0  392.71  4985.4  391.60  4985.8  391.10  4990.3  391.10
  4990.7  391.60  4997.9  391.75  5018.1  394.29  5028.4  394.73  5140.3  395.36
  5170.8  397.24  5231.8  396.51  5363.9  397.43  5374.1  397.02  5404.6  397.78
  5577.4  397.68  5658.7  398.56  5763.1  398.01  5875.0  399.33  5902.6  400.49
  5933.5  399.73  6055.1  399.54  6177.0  400.28  6238.0  399.90  6293.7  400.61
#Mann=3,-1,0
  4622.2    0.05       0  4985.4    0.05       0  4990.7    0.05       0
Bank Sta=4985.4,4990.7
Exp/Cntr=0.3,0.1

Type RM Length L Ch R = 1,58450,216,216,216
BEGIN DESCRIPTION:
Prairie Creek58450.35
END DESCRIPTION:
XS GIS Cut Line= 3
      2713293.10      6835136.39      2713181.35      6835363.31
      2712659.04      6836836.19
#Sta/Elev= 30
  4752.3  401.40  4782.5  400.65  4790.9  399.60  4821.9  399.37  4911.7  399.59
  4924.6  400.71  4934.2  400.13  4962.2  395.97  4979.1  392.73  4998.5  391.49
  4998.9  390.99  5003.4  390.99  5003.8  391.49  5013.4  393.28  5045.2  394.75
  5094.5  395.64  5428.8  396.66  5480.0  397.25  5490.9  398.19  5510.9  397.16
  5565.1  398.11  5639.7  397.51  5721.7  398.20  5796.6  397.80  5841.5  397.77
  6086.9  398.78  6106.3  399.84  6212.4  398.98  6503.2  399.56  6568.0  400.33
#Mann=5,-1,0
  4752.3    0.05       0  4998.5    0.05       0  5003.8    0.05       0
  5796.6    0.07       0  5841.5    0.05       0
Bank Sta=4998.5,5003.8
Exp/Cntr=0.3,0.1

Type RM Length L Ch R = 1,58234,246,246,246
BEGIN DESCRIPTION:
Prairie Creek58234.41
END DESCRIPTION:
XS GIS Cut Line= 3
      2713254.21      6835070.57      2712992.23      6835281.04
      2711695.69      6836436.73
#Sta/Elev= 30
  4666.2  401.92  4736.6  400.21  4807.0  399.56  4899.8  395.41  4914.2  394.18
  4943.0  393.99  4969.1  391.31  4969.5  390.81  4974.0  390.81  4974.4  391.31
  5002.2  391.96  5013.5  394.61  5027.7  395.09  5105.5  395.39  5133.9  394.54
  5172.1  394.79  5222.5  396.25  5417.3  396.30  5439.1  397.16  5452.7  396.55
  5509.3  396.97  5573.2  396.47  5770.4  397.15  5814.4  396.75  5884.7  398.03
  5913.1  396.61  5937.2  397.32  5948.3  396.83  6125.5  396.53  6739.1  398.12
#Mann=7,-1,0
  4666.2    0.05       0  4969.1    0.05       0  4974.4    0.05       0
  5172.1    0.07       0  5222.5    0.05       0  5770.4   0.063       0
  5937.2    0.05       0
Bank Sta=4969.1,4974.4
Exp/Cntr=0.3,0.1

Type RM Length L Ch R = 1,57988,290,290,290
BEGIN DESCRIPTION:
Mapping XS fe6308a3
END DESCRIPTION:
XS GIS Cut Line= 3
      2713106.31      6835063.49      2712795.99      6835138.63
      2711560.90      6835984.74
#Sta/Elev= 30
  4687.1  400.58  4944.6  393.87  4985.8  392.47  4995.4  390.77  4995.9  390.27
  5001.0  390.77  5036.9  394.13  5071.9  395.63  5087.7  394.37  5093.7  395.72
  5108.6  396.38  5123.6  395.23  5129.6  396.53  5159.4  395.19  5200.2  395.59
  5431.6  396.32  5512.1  397.00  5527.0  395.30  5554.1  396.23  5562.9  395.02
  5583.9  396.16  5618.4  395.83  5921.7  395.46  5993.4  396.26  6000.3  397.48
  6008.3  396.00  6376.0  396.50  6474.7  397.10  6493.0  398.23  6503.5  399.19
#Mann=8,-1,0
  4687.1    0.05       0  4995.4    0.05       0  5001.0    0.05       0
  5071.9    0.07       0  5200.2    0.05       0  5431.6   0.063       0
  5618.4    0.05       0  6493.0   0.063       0
Bank Sta=4995.4,5001
Exp/Cntr=0.3,0.1

Type RM Length L Ch R = 1,57698,230,230,230
BEGIN DESCRIPTION:
Prairie Creek57698.1
END DESCRIPTION:
XS GIS Cut Line= 4
      2713344.22      6835015.16      2712541.61      6835031.36
      2711722.57      6834995.26      2710721.49      6834955.01
#Sta/Elev= 30
  4201.5  403.64  4549.8  398.98  4609.8  396.51  4749.8  394.85  4809.8  393.21
  4949.9  392.50  5037.1  389.66  5037.6  389.16  5042.7  389.66  5061.3  391.48
  5080.0  393.41  5110.0  394.39  5120.0  395.37  5130.5  393.55  5150.0  394.64
  5170.0  393.18  5310.2  395.46  5460.3  393.52  5500.4  394.02  5600.5  393.49
  5690.5  394.44  5819.9  393.36  6099.3  393.89  6231.0  394.78  6251.0  394.03
  6411.2  392.87  6691.4  394.13  6701.4  393.40  6741.4  394.48  6826.0  394.54
#Mann=5,-1,0
  4201.5    0.05       0  5037.1    0.05       0  5042.7    0.05       0
  5061.3   0.063       0  6099.3    0.05       0
Bank Sta=5037.1,5042.7
Exp/Cntr=0.3,0.1

Type RM Length L Ch R = 1,57468,649,649,649
BEGIN DESCRIPTION:
Prairie Creek57468.36
END DESCRIPTION:
XS GIS Cut Line= 4
      2713276.92      6834875.07      2712389.28      6834882.40
      2711373.30      6834848.71      2710750.94      6834820.60
#Sta/Elev= 30
  4120.9  405.66  4151.8  404.56  4221.8  403.79  4241.8  402.66  4371.8  401.28
  4411.8  399.65  4481.8  398.22  4741.2  394.61  4841.8  393.10  4921.8  393.78
  4951.8  392.84  4969.0  390.46  4969.5  389.96  4974.6  390.46  5001.9  392.45
  5161.9  393.40  5199.3  394.42  5262.0  393.52  5342.0  393.84  5422.1  392.74
  5632.2  391.80  5782.3  392.41  6002.4  391.18  6021.3  391.82  6292.7  391.44
  6332.7  392.38  6412.8  391.95  6452.8  393.11  6601.4  394.03  6648.1  394.04
#Mann=5,-1,0
  4120.9   0.063       0  4741.2    0.05       0  4969.0    0.05       0
  4974.6    0.05       0  6601.4   0.063       0
Bank Sta=4969,4974.6
Exp/Cntr=0.3,0.1

Type RM Length L Ch R = 1,56819,709,709,709
BEGIN DESCRIPTION:
Mapping XS 7407bad1
END DESCRIPTION:
XS GIS Cut Line= 3
      2712201.43      6834229.58      2711915.61      6834520.86
      2710801.50      6834793.20
#Sta/Elev= 30
  4606.1  399.79  4646.3  399.07  4660.5  399.75  4702.9  397.68  4808.9  394.97
  4893.8  390.48  4971.6  391.00  4985.8  390.38  4992.8  388.99  5006.9  388.15
  5016.6  388.58  5032.5  392.40  5044.7  392.43  5209.4  391.08  5281.4  391.51
  5459.3  390.64  5549.1  389.51  5579.1  390.26  5628.5  387.96  5629.0  387.46
  5634.4  387.96  5652.0  388.38  5682.9  391.17  5693.2  391.36  5868.2  389.28
  5880.9  389.69  5899.1  391.55  5950.6  390.52  6022.6  392.21  6161.1  393.99
#Mann=3,-1,0
  4606.1    0.05       0  5628.5    0.05       0  5634.4    0.05       0
Bank Sta=5628.5,5634.4
Exp/Cntr=0.3,0.1

Type RM Length L Ch R = 1,56110,656,656,656
BEGIN DESCRIPTION:
Prairie Creek56110.24
END DESCRIPTION:
XS GIS Cut Line= 4
      2711763.42      6834008.56      2711428.84      6834374.94
      2710994.60      6834666.32      2710639.60      6834828.98
#Sta/Elev= 30
  4510.8  397.90  4553.4  398.04  4567.6  397.01  4708.8  394.01  4900.0  392.32
  4914.2  390.28  4928.4  390.24  4949.3  388.33  4956.8  389.07  4963.5  387.17
  4985.1  387.98  5002.4  386.30  5002.9  385.80  5008.4  386.30  5021.6  386.76
  5027.6  388.06  5057.6  388.87  5063.6  390.06  5165.7  389.12  5192.7  389.92
  5279.7  389.64  5315.7  387.93  5366.7  387.52  5417.7  388.78  5510.8  388.34
  5525.8  390.54  5539.4  391.04  5759.4  393.78  5855.5  393.77  5920.4  394.35
#Mann=4,-1,0
  4510.8    0.05       0  5002.4    0.05       0  5008.4    0.05       0
  5855.5   0.063       0
Bank Sta=5002.4,5008.4
Exp/Cntr=0.3,0.1

Type RM Length L Ch R = 1,55454,614,614,614
BEGIN DESCRIPTION:
Prairie Creek55453.5
END DESCRIPTION:
XS GIS Cut Line= 3
      2711330.72      6833655.75      2710833.73      6834376.90
      2710560.03      6834821.01
#Sta/Elev= 30
  4129.5  395.45  4186.2  394.54  4281.6  394.34  4302.5  393.33  4410.1  392.05
  4460.8  392.29  4481.7  391.22  4517.6  390.64  4597.4  390.26  4610.2  390.71
  4711.7  388.81  4798.2  389.19  4913.1  387.84  4962.5  386.89  4977.4  383.70
  4989.0  383.69  4989.5  383.19  4995.0  383.19  4995.5  383.69  4998.4  385.03
  5007.9  383.96  5013.3  387.01  5028.7  387.30  5034.5  389.82  5049.9  390.62
  5080.6  390.26  5239.2  392.66  5336.2  393.08  5492.2  393.63  5527.0  393.87
#Mann=5,-1,0
  4129.5    0.05       0  4989.0    0.05       0  4995.5    0.05       0
  5336.2   0.035       0  5492.2   0.063       0
Bank Sta=4989,4995.5
Exp/Cntr=0.3,0.1

Type RM Length L Ch R = 1,54840,758,758,758
BEGIN DESCRIPTION:
Prairie Creek54839.6
END DESCRIPTION:
XS GIS Cut Line= 3
      2710779.50      6833087.26      2710541.99      6834027.33
      2710398.19      6834725.37
#Sta/Elev= 30
  4047.3  393.65  4133.7  392.35  4207.7  392.45  4298.7  390.76  4366.7  390.96
  4731.0  387.14  4793.8  387.16  4854.1  388.18  4900.3  387.24  4969.1  387.35
  4977.2  387.09  4982.4  386.08  4989.7  386.04  5000.1  383.74  5007.1  381.16
  5007.6  380.66  5013.2  380.66  5013.7  381.16  5016.2  383.31  5019.4  383.31
  5023.8  385.93  5051.3  385.20  5074.1  386.07  5081.9  387.18  5119.3  387.90
  5124.4  388.52  5204.4  389.11  5275.9  391.07  5493.8  392.23  5729.6  393.66
#Mann=4,-1,0
  4047.3    0.05       0  5007.1    0.05       0  5013.7    0.05       0
  5493.8   0.035       0
Bank Sta=5007.1,5013.7
Exp/Cntr=0.3,0.1

Type RM Length L Ch R = 1,54082,172,172,172
BEGIN DESCRIPTION:
Prairie Creek54082.16
END DESCRIPTION:
XS GIS Cut Line= 3
      2710138.86      6832766.02      2710108.06      6833534.24
      2710110.50      6834583.70
#Sta/Elev= 30
  4254.2  390.50  4499.4  389.39  4519.4  388.64  4697.3  387.43  4702.3  387.86
  4709.5  387.43  4769.6  387.04  4869.7  386.80  4939.7  385.26  4969.8  385.13
  4989.8  383.75  4999.8  381.94  5009.8  380.69  5015.4  380.60  5015.9  380.10
  5021.9  380.10  5022.4  380.60  5029.8  381.37  5039.8  383.78  5069.8  386.17
  5229.8  387.21  5269.8  388.06  5309.8  388.21  5329.8  388.69  5349.8  388.35
  5629.8  390.20  5789.8  390.39  5939.8  392.20  6039.8  392.31  6072.5  393.08
#Mann=3,-1,0
  4254.2   0.063       0  5015.4   0.063       0  5022.4   0.063       0
Bank Sta=5015.4,5022.4
Exp/Cntr=0.3,0.1

Type RM Length L Ch R = 1,53910,388,388,388
BEGIN DESCRIPTION:
Prairie Creek53909.84
END DESCRIPTION:
XS GIS Cut Line= 3
      2709954.41      6832735.81      2709936.36      6833525.12
      2709916.92      6834567.42
#Sta/Elev= 30
  4224.6  390.34  4399.8  390.27  4429.8  389.42  4634.0  388.48  4729.5  388.27
  4765.4  387.56  4779.9  387.67  4813.0  384.74  4970.0  386.27  4990.0  383.22
  5000.0  380.55  5006.1  380.37  5006.6  379.87  5013.1  380.37  5020.0  380.80
  5030.0  383.52  5040.0  384.94  5052.9  385.25  5110.0  385.17  5140.0  386.71
  5240.0  388.42  5250.0  389.49  5285.8  389.33  5350.1  390.63  5481.6  390.07
  5657.2  391.68  5800.4  391.46  5849.4  391.42  5930.2  392.78  6056.6  392.37
#Mann=12,-1,0
  4224.6   0.063       0  4634.0   0.035       0  4729.5   0.063       0
  4765.4   0.035       0  5006.1   0.035       0  5013.1   0.035       0
  5052.9   0.063       0  5285.8   0.035       0  5481.6   0.063       0
  5657.2   0.035       0  5800.4   0.063       0  5849.4   0.035       0
Bank Sta=5006.1,5013.1
Exp/Cntr=0.3,0.1

Type RM Length L Ch R = 1,53522,686,686,686
BEGIN DESCRIPTION:
Prairie Creek53521.9
END DESCRIPTION:
XS GIS Cut Line= 3
      2709711.32      6832740.82      2709619.67      6833375.19
      2709512.75      6834035.13
#Sta/Elev= 30
  4370.2  389.07  4400.7  388.39  4481.5  389.43  4514.6  388.26  4572.5  388.58
  4655.3  387.59  4725.6  385.18  4754.3  386.47  4784.6  385.17  4795.9  383.83
  4835.2  383.10  4866.2  383.23  4905.9  384.62  4936.6  384.22  4976.6  384.86
  4996.8  382.62  5001.9  380.89  5003.0  378.57  5003.5  378.07  5010.1  378.57
  5017.0  378.76  5027.2  382.28  5037.3  384.19  5060.4  384.99  5148.7  385.49
  5192.4  387.93  5351.3  388.16  5382.4  389.44  5448.1  389.54  5679.7  390.28
#Mann=5,-1,0
  4370.2    0.05       0  5003.0    0.05       0  5010.1    0.05       0
  5060.4   0.063       0  5448.1   0.094       0
Bank Sta=5003,5010.1
Exp/Cntr=0.3,0.1

Type RM Length L Ch R = 1,52836,971,971,971
BEGIN DESCRIPTION:
Prairie Creek52835.95
END DESCRIPTION:
XS GIS Cut Line= 3
      2709642.02      6832717.65      2709168.54      6833022.86
      2708426.11      6833360.93
#Sta/Elev= 30
  4442.6  388.38  4565.8  386.14  4659.5  386.77  4738.1  382.97  4789.5  385.26
  4810.7  382.66  4854.3  383.00  4868.1  384.16  4898.4  382.83  4971.1  382.57
  4998.1  380.45  5004.5  377.57  5016.0  376.45  5016.5  375.95  5023.5  376.45
  5030.7  378.05  5036.9  382.14  5042.4  382.81  5106.1  382.51  5249.9  384.16
  5272.4  382.76  5282.1  383.65  5372.3  386.34  5445.3  385.03  5548.5  387.24
  5580.1  386.81  5594.6  388.01  5624.0  388.40  5669.3  389.41  5821.7  387.91
#Mann=6,-1,0
  4442.6    0.05       0  5016.0    0.05       0  5023.5    0.05       0
  5282.1   0.035       0  5372.3   0.063       0  5624.0    0.05       0
Bank Sta=5016,5023.5
Exp/Cntr=0.3,0.1

Type RM Length L Ch R = 1,51865,221,221,221
BEGIN DESCRIPTION:
Prairie Creek51864.89
END DESCRIPTION:
XS GIS Cut Line= 3
      2709566.17      6832663.94      2708618.48      6832659.61
      2708056.65      6832651.12
#Sta/Elev= 30
  4055.8  387.50  4326.0  385.71  4396.0  386.24  4446.0  384.44  4466.0  384.92
  4496.0  384.49  4516.0  383.53  4576.0  382.35  4616.0  382.62  4636.0  383.36
  4746.0  382.44  4846.0  382.84  4886.0  381.45  4926.0  382.43  4946.0  381.97
  4976.0  380.09  5016.0  380.49  5026.0  377.32  5032.0  374.33  5032.5  373.83
  5039.4  373.83  5039.9  374.33  5046.0  378.12  5056.0  380.49  5096.0  382.35
  5136.0  382.14  5176.0  383.89  5226.0  385.13  5296.0  384.56  5565.4  386.23
#Mann=3,-1,0
  4055.8    0.05       0  5032.0    0.05       0  5039.9    0.05       0
Bank Sta=5032,5039.9
Exp/Cntr=0.3,0.1

Type RM Length L Ch R = 1,51644,527,527,527
BEGIN DESCRIPTION:
Prairie Creek51643.94
END DESCRIPTION:
XS GIS Cut Line= 3
      2709511.07      6832502.50      2708519.33      6832497.16
      2708052.63      6832503.83
#Sta/Elev= 30
  4015.3  387.67  4090.4  386.65  4180.4  386.68  4240.4  385.47  4380.4  385.42
  4480.4  383.86  4530.4  385.45  4560.4  383.85  4620.4  384.03  4650.4  380.35
  4680.4  379.57  4700.4  379.83  4730.4  381.90  4760.4  383.03  4820.4  381.26
  4880.4  381.64  4900.4  380.59  4950.4  379.77  4990.4  380.31  5002.3  376.18
  5002.8  375.68  5009.7  375.68  5010.2  376.18  5020.4  379.83  5030.4  381.18
  5050.4  382.68  5080.4  383.86  5120.4  383.45  5280.4  383.93  5473.8  385.70
#Mann=3,-1,0
  4015.3    0.05       0  5002.3    0.05       0  5010.2    0.05       0
Bank Sta=5002.3,5010.2
Exp/Cntr=0.3,0.1

Type RM Length L Ch R = 1,51117,448,448,448
BEGIN DESCRIPTION:
Prairie Creek51117.39
END DESCRIPTION:
XS GIS Cut Line= 3
      2709270.04      6832116.01      2708819.77      6832209.62
      2708114.84      6832353.72
#Sta/Elev= 30
  4546.9  387.19  4622.5  386.30  4653.2  386.68  4683.8  385.71  4775.7  384.92
  4847.2  384.71  4867.7  385.27  4877.9  384.36  4937.0  383.03  4959.6  381.43
  4980.0  378.52  4983.1  373.86  4983.6  373.36  4990.5  373.36  4991.0  373.86
  5000.4  377.99  5037.4  379.07  5071.9  379.32  5087.9  378.77  5138.4  380.02
  5265.8  380.88  5296.4  380.10  5347.5  381.57  5398.5  381.87  5436.2  383.28
  5480.2  382.85  5486.6  383.27  5521.0  383.11  5537.1  383.86  5726.3  384.93
#Mann=3,-1,0
  4546.9    0.05       0  4983.1    0.05       0  4991.0    0.05       0
Bank Sta=4983.1,4991
Exp/Cntr=0.3,0.1

Type RM Length L Ch R = 1,50669,292,292,292
BEGIN DESCRIPTION:
Prairie Creek50668.81
END DESCRIPTION:
XS GIS Cut Line= 3
      2709041.78      6831761.28      2708624.35      6831893.76
      2708162.02      6832061.60
#Sta/Elev= 30
  4563.8  384.69  4679.3  383.67  4685.3  382.96  4711.6  382.01  4758.7  381.93
  4776.1  380.81  4863.6  379.79  4872.9  380.49  4895.1  379.54  4905.2  378.53
  4958.1  378.18  4968.5  377.02  4970.9  374.18  4971.4  373.68  4978.4  373.68
  4978.9  374.18  4980.2  375.36  4989.5  374.27  4998.3  378.39  5006.8  379.29
  5012.1  375.28  5021.3  379.41  5042.7  380.83  5053.2  380.13  5074.5  379.86
  5106.4  380.68  5202.1  380.86  5297.0  382.24  5358.2  382.01  5493.6  383.77
#Mann=3,-1,0
  4563.8    0.05       0  4970.9    0.05       0  4978.9    0.05       0
Bank Sta=4970.9,4978.9
Exp/Cntr=0.3,0.1

Type RM Length L Ch R = 1,50377,199,199,199
BEGIN DESCRIPTION:
Prairie Creek50376.97
END DESCRIPTION:
XS GIS Cut Line= 3
      2709051.09      6831546.76      2708676.92      6831650.79
      2708139.64      6831814.72
#Sta/Elev= 30
  4611.5  384.47  4710.2  383.79  4741.3  382.75  4803.6  383.62  4831.1  381.94
  4886.6  379.93  4904.8  378.33  4910.0  379.16  4917.8  377.92  4928.2  377.22
  4944.2  377.31  4949.4  376.65  4969.7  377.62  5003.0  377.72  5007.3  373.98
  5007.8  373.48  5014.8  373.48  5015.3  373.98  5022.3  377.30  5074.0  378.14
  5094.9  379.74  5251.8  379.54  5322.9  380.21  5345.8  380.95  5366.8  380.52
  5426.6  381.68  5459.4  381.28  5471.3  381.99  5502.7  381.28  5561.6  381.48
#Mann=3,-1,0
  4611.5    0.05       0  5007.3    0.05       0  5015.3    0.05       0
Bank Sta=5007.3,5015.3
Exp/Cntr=0.3,0.1

Type RM Length L Ch R = 1,50178,230,230,230
BEGIN DESCRIPTION:
Prairie Creek50177.8
END DESCRIPTION:
XS GIS Cut Line= 3
      2709017.15      6831360.68      2708591.20      6831479.12
      2707831.96      6831743.61
#Sta/Elev= 30
  4560.6  384.04  4603.3  383.80  4624.1  384.15  4652.6  383.20  4770.8  382.42
  4805.1  381.62  4844.5  380.15  4873.2  378.02  4904.3  377.11  4925.1  375.94
  4945.8  375.85  4952.4  374.59  4957.6  372.77  4962.6  372.71  4963.1  372.21
  4970.1  372.21  4970.6  372.71  4986.6  376.30  5023.9  377.02  5061.2  379.38
  5220.0  379.23  5251.8  379.97  5315.3  379.80  5368.3  380.83  5386.3  380.45
  5453.7  380.84  5479.5  380.43  5536.4  380.58  5738.9  382.87  5806.7  384.05
#Mann=3,-1,0
  4560.6    0.05       0  4962.6    0.05       0  4970.6    0.05       0
Bank Sta=4962.6,4970.6
Exp/Cntr=0.3,0.1

Type RM Length L Ch R = 1,49948,174,174,174
BEGIN DESCRIPTION:
Prairie Creek49948.03
END DESCRIPTION:
XS GIS Cut Line= 3
      2708655.65      6831229.50      2708438.88      6831328.44
      2707894.38      6831585.70
#Sta/Elev= 30
  4764.9  382.54  4775.3  382.95  4786.5  382.21  4803.8  378.82  4819.5  377.67
  4826.9  376.30  4855.4  376.52  4863.5  374.81  4872.9  374.13  4878.4  374.60
  4885.4  373.95  4924.5  374.27  4930.0  375.46  4953.0  374.67  4962.4  375.49
  4970.6  375.06  4976.1  375.90  4984.4  373.92  4989.6  371.88  4990.1  371.38
  4997.1  371.38  4997.6  371.88  4999.1  374.97  5009.2  375.41  5016.4  377.02
  5028.5  378.30  5050.6  378.87  5346.2  379.39  5374.5  380.15  5605.4  382.22
#Mann=4,-1,0
  4764.9    0.16       0  4989.6    0.07       0  4997.6    0.16       0
  5009.2    0.05       0
Bank Sta=4989.6,4997.6
Exp/Cntr=0.3,0.1

Type RM Length L Ch R = 1,49774,261,261,261
BEGIN DESCRIPTION:
Prairie Creek49773.63
END DESCRIPTION:
XS GIS Cut Line= 3
      2708797.38      6831040.83      2708374.13      6831173.15
      2707950.01      6831320.70
#Sta/Elev= 30
  4558.0  381.81  4664.2  380.90  4775.3  378.95  4821.4  379.19  4840.3  378.45
  4905.2  377.15  4910.4  376.56  4942.9  376.20  4980.6  377.27  4985.0  371.89
  4985.5  371.39  4992.6  371.39  4993.1  371.89  4997.8  373.78  5001.4  373.78
  5007.4  376.90  5012.7  376.23  5020.6  376.88  5031.2  376.89  5074.9  378.40
  5115.9  378.57  5147.7  378.25  5157.6  379.38  5162.9  378.25  5188.7  378.80
  5200.6  378.46  5211.2  378.69  5243.0  377.76  5313.1  379.49  5450.5  381.01
#Mann=3,-1,0
  4558.0    0.05       0  4985.0    0.05       0  4993.1    0.05       0
Bank Sta=4985,4993.1
Exp/Cntr=0.3,0.1

Type RM Length L Ch R = 1,49513,301,301,301
BEGIN DESCRIPTION:
Prairie Creek49513.42
END DESCRIPTION:
XS GIS Cut Line= 3
      2708712.71      6830825.86      2708426.74      6830928.45
      2707925.52      6831128.28
#Sta/Elev= 30
  4695.4  383.07  4721.9  383.13  4830.0  381.22  4870.4  378.98  4931.8  376.78
  4946.9  377.49  4968.1  375.77  4978.8  372.50  4984.0  371.97  4984.5  371.47
  4991.6  371.47  4992.1  371.97  4993.3  372.39  4997.0  375.15  5023.3  376.57
  5032.3  375.87  5071.8  376.10  5125.7  377.74  5155.4  378.09  5238.9  377.18
  5247.6  376.63  5257.8  377.76  5263.2  377.00  5269.1  376.95  5292.8  378.02
  5311.7  377.93  5333.7  376.86  5365.6  377.30  5409.1  378.79  5538.8  379.82
#Mann=3,-1,0
  4695.4    0.05       0  4984.0    0.05       0  4992.1    0.05       0
Bank Sta=4984,4992.1
Exp/Cntr=0.3,0.1

Type RM Length L Ch R = 1,49212,226,226,226
BEGIN DESCRIPTION:
Prairie Creek49212.37
END DESCRIPTION:
XS GIS Cut Line= 3
      2708571.74      6830540.78      2708228.50      6830706.13
      2707816.79      6830909.75
#Sta/Elev= 30
  4619.0  381.61  4721.5  380.61  4727.0  379.92  4744.1  379.88  4789.3  378.07
  4879.8  376.29  4891.8  375.48  4925.0  374.43  4930.6  374.66  4947.3  374.00
  4958.8  374.23  4971.7  371.57  4972.2  371.07  4979.5  371.07  4980.0  371.57
  4991.7  375.22  5004.2  375.71  5020.9  374.70  5093.8  376.84  5110.6  376.58
  5161.1  377.32  5200.4  376.25  5228.4  376.22  5237.1  375.82  5267.7  376.48
  5273.2  375.96  5290.1  376.83  5379.8  378.04  5437.9  379.50  5459.3  379.32
#Mann=3,-1,0
  4619.0    0.05       0  4971.7    0.05       0  4980.0    0.05       0
Bank Sta=4971.7,4980
Exp/Cntr=0.3,0.1

Type RM Length L Ch R = 1,48986,264,264,264
BEGIN DESCRIPTION:
Prairie Creek48986.31
END DESCRIPTION:
XS GIS Cut Line= 3
      2708508.11      6830341.04      2708173.95      6830497.04
      2707743.71      6830756.69
#Sta/Elev= 30
  4632.7  380.67  4688.2  379.77  4693.7  380.42  4701.2  379.90  4711.1  379.64
  4716.6  379.95  4733.9  379.24  4739.4  379.55  4762.3  378.93  4790.7  378.78
  4866.8  376.09  4922.0  375.21  4927.8  374.44  4979.0  374.38  4988.2  373.74
  4992.2  370.69  4992.7  370.19  5000.0  370.19  5000.5  370.69  5010.8  373.70
  5017.7  375.15  5033.2  375.80  5075.9  374.82  5104.2  376.24  5127.6  376.57
  5155.5  376.64  5171.0  375.85  5244.4  375.79  5404.0  378.01  5504.0  378.67
#Mann=3,-1,0
  4632.7    0.05       0  4992.2    0.05       0  5000.5    0.05       0
Bank Sta=4992.2,5000.5
Exp/Cntr=0.3,0.1

Type RM Length L Ch R = 1,48722,257,257,257
BEGIN DESCRIPTION:
Mapping XS 46c28997
END DESCRIPTION:
XS GIS Cut Line= 3
      2708431.89      6830084.74      2708216.39      6830256.44
      2707627.82      6830686.19
#Sta/Elev= 30
  4737.4  380.86  4852.7  379.19  4867.1  377.95  4887.9  378.58  4895.9  376.91
  4902.3  377.91  4910.4  374.96  4916.7  376.37  4931.2  372.38  4937.6  373.96
  4945.6  372.73  4952.0  373.98  4960.0  373.12  4966.4  375.79  4974.4  375.50
  4995.2  371.48  5001.6  371.77  5005.5  369.60  5006.0  369.10  5013.8  369.60
  5024.4  371.62  5030.6  370.39  5051.4  374.36  5066.1  375.12  5181.2  374.33
  5266.9  376.48  5402.8  375.55  5509.4  378.27  5553.4  377.49  5741.7  378.78
#Mann=3,-1,0
  4737.4    0.05       0  5005.5    0.05       0  5013.8    0.05       0
Bank Sta=5005.5,5013.8
Exp/Cntr=0.3,0.1

Type RM Length L Ch R = 1,48465,242,242,242
BEGIN DESCRIPTION:
Prairie Creek48497.72
END DESCRIPTION:
XS GIS Cut Line= 3
      2708211.48      6829912.17      2708038.13      6830108.63
      2707643.13      6830617.39
#Sta/Elev= 30
  4738.0  378.60  4812.0  378.07  4875.6  375.85  4939.2  375.78  4946.7  374.54
  4962.5  374.42  4974.4  374.30  4981.9  374.01  4989.4  371.72  4996.1  371.98
  4998.2  370.31  5004.7  370.31  5010.5  371.71  5027.1  368.69  5027.6  368.19
  5035.5  368.69  5060.3  372.32  5066.6  371.96  5074.7  373.78  5081.1  373.28
  5089.2  374.48  5153.5  375.84  5167.6  375.25  5195.1  375.93  5209.6  375.36
  5294.7  376.00  5381.6  375.15  5431.4  376.90  5458.8  376.52  5644.1  378.18
#Mann=5,-1,0
  4738.0    0.05       0  4962.5    0.16       0  4974.4    0.05       0
  5027.1    0.05       0  5035.5    0.05       0
Bank Sta=5027.1,5035.5
Exp/Cntr=0.3,0.1

Type RM Length L Ch R = 1,48223,482,482,482
BEGIN DESCRIPTION:
Mapping XS 16bc51e6
END DESCRIPTION:
XS GIS Cut Line= 3
      2708193.66      6829823.45      2707900.11      6829936.25
      2707482.25      6829991.66
#Sta/Elev= 30
  4686.7  377.91  4769.9  377.14  4781.7  377.55  4823.5  376.06  4885.7  375.96
  4891.0  375.83  4898.5  374.55  4921.0  374.55  4940.1  373.74  4970.3  373.82
  4975.7  374.25  5015.4  373.30  5025.5  371.38  5031.4  368.11  5031.9  367.61
  5039.3  367.61  5039.8  368.11  5045.7  368.46  5055.8  371.70  5065.8  371.41
  5086.0  373.79  5126.4  373.34  5167.7  374.28  5197.0  375.09  5247.4  374.70
  5277.7  375.60  5308.3  377.32  5348.3  376.79  5398.7  378.40  5422.7  377.99
#Mann=5,-1,0
  4686.7    0.05       0  4940.1    0.16       0  5031.4    0.07       0
  5039.8    0.16       0  5167.7    0.05       0
Bank Sta=5031.4,5039.8
Exp/Cntr=0.3,0.1

Type RM Length L Ch R = 1,47741,397,397,397
BEGIN DESCRIPTION:
Prairie Creek48117.07
END DESCRIPTION:
XS GIS Cut Line= 3
      2708233.98      6829699.69      2707645.14      6829581.42
      2707483.59      6829935.17
#Sta/Elev= 30
  4399.4  378.06  4478.9  377.47  4499.3  376.14  4550.3  375.42  4693.1  374.56
  4733.9  375.03  4754.3  374.19  4764.5  374.47  4776.7  373.58  4883.2  372.94
  4929.4  373.44  4937.9  372.66  4975.2  372.02  5007.5  368.90  5008.7  367.29
  5009.2  366.79  5016.7  366.79  5017.2  367.29  5021.5  369.41  5030.5  372.04
  5036.0  372.38  5043.5  371.64  5059.1  372.65  5098.5  371.86  5133.6  374.08
  5175.6  375.11  5225.8  376.09  5231.3  377.17  5263.4  376.65  5388.9  378.33
#Mann=5,-1,0
  4399.4    0.05       0  4883.2    0.16       0  5008.7    0.07       0
  5017.2    0.16       0  5175.6    0.05       0
Bank Sta=5008.7,5017.2
Exp/Cntr=0.3,0.1

Type RM Length L Ch R = 1,47344,347,347,347
BEGIN DESCRIPTION:
Prairie Creek47344.16
END DESCRIPTION:
XS GIS Cut Line= 3
      2707520.93      6828764.48      2707491.31      6829290.22
      2707463.06      6829885.27
#Sta/Elev= 30
  4486.8  380.69  4533.4  380.09  4573.5  378.50  4583.5  377.41  4603.5  372.44
  4627.7  371.51  4907.8  372.94  4974.1  372.26  4984.1  368.40  4988.4  364.55
  4988.9  364.05  4999.9  364.55  5004.1  364.63  5011.3  366.56  5016.3  366.56
  5019.6  370.34  5024.6  371.80  5034.2  372.49  5088.5  372.03  5124.3  372.79
  5164.3  371.35  5224.4  371.25  5284.5  373.59  5314.5  375.49  5349.0  375.24
  5394.6  375.25  5445.7  376.55  5467.7  377.82  5534.7  376.96  5609.1  378.55
#Mann=8,-1,0
  4486.8    0.05       0  4627.7    0.07       0  4907.8   0.035       0
  4988.4   0.035       0  4999.9   0.035       0  5088.5    0.16       0
  5349.0    0.05       0  5467.7    0.16       0
Bank Sta=4988.4,4999.9
Exp/Cntr=0.3,0.1

Type RM Length L Ch R = 1,46997,384,384,384
BEGIN DESCRIPTION:
Prairie Creek46965.74
END DESCRIPTION:
XS GIS Cut Line= 3
      2707190.47      6828459.70      2707185.59      6829159.79
      2707384.36      6829855.76
#Sta/Elev= 30
  4299.9  378.29  4371.2  377.88  4431.2  375.82  4491.2  375.56  4621.2  373.42
  4661.2  373.58  4731.2  372.17  4811.2  371.40  4901.2  371.88  4911.2  371.55
  4941.2  368.56  4951.2  365.10  4965.5  363.80  4966.0  363.30  4976.5  363.30
  4977.0  363.80  4991.2  364.89  4998.1  367.37  5003.2  367.37  5011.7  369.16
  5057.3  368.87  5084.5  369.90  5130.1  369.35  5136.5  370.01  5163.9  369.41
  5178.1  370.60  5188.5  370.32  5202.9  371.21  5323.7  371.09  5723.8  376.07
#Mann=3,-1,0
  4299.9    0.05       0  4965.5    0.05       0  4977.0    0.05       0
Bank Sta=4965.5,4977
Exp/Cntr=0.3,0.1

Type RM Length L Ch R = 1,46613,251,251,251
BEGIN DESCRIPTION:
Prairie Creek46612.85
END DESCRIPTION:
XS GIS Cut Line= 3
      2706916.49      6828429.42      2706874.97      6828961.87
      2706791.03      6830196.26
#Sta/Elev= 30
  4472.1  379.22  4664.3  373.07  4724.4  372.01  4799.8  371.93  4874.9  370.77
  4965.2  371.16  4985.2  365.51  4989.5  363.65  4990.0  363.15  5000.5  363.15
  5001.0  363.65  5015.3  364.02  5025.3  365.28  5035.4  367.94  5055.4  371.27
  5062.6  371.82  5145.6  370.44  5165.9  370.67  5195.7  370.33  5211.5  371.68
  5235.8  369.64  5263.9  369.63  5672.7  369.50  5841.0  369.47  5949.8  369.45
  6047.8  369.44  6067.7  369.81  6087.8  373.83  6099.6  374.53  6243.4  376.24
#Mann=9,-1,0
  4472.1    0.05       0  4989.5    0.05       0  5001.0    0.05       0
  5165.9   0.035       0  5263.9   0.033       0  5672.7   0.035       0
  5841.0   0.033       0  5949.8   0.035       0  6047.8    0.05       0
Bank Sta=4989.5,5001
Exp/Cntr=0.3,0.1

Type RM Length L Ch R = 1,46362,320,320,320
BEGIN DESCRIPTION:
Prairie Creek46219.55
END DESCRIPTION:
XS GIS Cut Line= 4
      2706687.09      6828365.19      2706659.51      6828843.90
      2706571.23      6829971.52      2706204.79      6830702.43
#Sta/Elev= 30
  4520.5  379.29  4816.8  370.65  4967.1  370.27  4973.1  367.51  4987.1  364.58
  5011.4  363.38  5011.9  362.88  5023.0  363.38  5057.3  370.77  5097.4  371.51
  5137.5  370.73  5177.6  371.82  5272.8  370.34  5298.0  370.99  5318.1  369.62
  5370.8  369.65  5807.8  369.69  5820.2  369.70  6057.1  369.72  6157.6  369.76
  6164.1  370.57  6172.9  374.07  6178.5  374.19  6195.3  377.51  6217.6  378.29
  6418.7  378.17  6491.3  376.60  6692.4  378.09  6843.2  376.91  6948.7  377.55
#Mann=9,-1,0
  4520.5    0.05       0  5011.4    0.05       0  5023.0    0.05       0
  5272.8   0.035       0  5370.8   0.033       0  5807.8   0.035       0
  5820.2   0.033       0  6057.1   0.035       0  6157.6    0.05       0
Bank Sta=5011.4,5023
Exp/Cntr=0.3,0.1

Type RM Length L Ch R = 1,46042,311,311,311
BEGIN DESCRIPTION:
Prairie Creek46042.043
END DESCRIPTION:
XS GIS Cut Line= 3
      2706402.79      6828337.52      2706385.78      6828721.54
      2706023.15      6830336.84
#Sta/Elev= 30
  4615.6  376.62  4655.1  375.17  4660.1  375.76  4839.3  372.13  4883.2  371.01
  4919.4  369.04  4969.4  368.29  4989.5  365.04  4997.2  362.97  5003.8  362.47
  5004.3  361.97  5015.5  362.47  5023.4  362.90  5060.9  370.27  5066.8  370.66
  5153.2  371.29  5194.2  369.09  5214.7  369.18  5235.2  370.78  5307.5  371.23
  5358.2  369.42  6294.2  369.62  6346.5  369.60  6352.3  371.04  6362.5  371.12
  6383.0  375.02  6413.8  375.80  6536.8  377.60  6578.5  376.96  6655.5  377.44
#Mann=5,-1,0
  4615.6    0.05       0  5003.8    0.05       0  5015.5    0.05       0
  5307.5   0.033       0  6294.2    0.05       0
Bank Sta=5003.8,5015.5
Exp/Cntr=0.3,0.1

Type RM Length L Ch R = 1,45731,319,319,319
BEGIN DESCRIPTION:
Mapping XS b5c9ac5b
END DESCRIPTION:
XS GIS Cut Line= 3
      2705991.65      6828186.58      2706095.26      6828670.32
      2706011.80      6830272.03
#Sta/Elev= 30
  4514.9  376.31  4621.7  374.72  4788.3  374.03  4856.9  373.69  4893.2  371.34
  4898.4  371.53  4928.5  369.95  4942.7  368.75  4959.2  366.29  4979.6  362.31
  4980.7  361.27  4981.2  360.77  4992.8  360.77  4993.3  361.27  5000.1  361.46
  5007.4  363.48  5020.3  364.13  5036.4  366.76  5050.4  368.84  5070.4  369.79
  5160.5  370.34  5420.9  369.48  5611.1  369.49  5651.2  370.16  6323.6  369.65
  6392.2  369.65  6402.2  373.98  6422.2  375.80  6562.4  377.30  6613.5  376.82
#Mann=6,-1,0
  4514.9   0.063       0  4788.3    0.05       0  4980.7    0.05       0
  4993.3    0.05       0  5036.4   0.033       0  6323.6    0.05       0
Bank Sta=4980.7,4993.3
Exp/Cntr=0.3,0.1

Type RM Length L Ch R = 1,45412,431,431,431
BEGIN DESCRIPTION:
Prairie Creek45411.66
END DESCRIPTION:
XS GIS Cut Line= 3
      2705795.50      6828224.08      2705790.31      6828613.62
      2705757.38      6830223.41
#Sta/Elev= 30
  4612.4  373.91  4679.3  373.27  4739.3  373.31  4867.8  371.79  4969.3  368.56
  4979.3  367.13  4989.3  363.18  4991.8  360.97  4992.3  360.47  5004.5  360.97
  5019.4  361.89  5049.4  366.86  5069.4  366.56  5099.4  370.31  5133.4  369.65
  5219.4  369.42  5259.4  370.31  5669.5  369.47  5759.5  370.10  5819.5  369.67
  5849.5  370.58  5889.5  369.99  6189.6  369.85  6364.9  370.50  6462.7  369.78
  6469.7  369.82  6479.7  373.65  6489.7  375.70  6589.7  377.78  6612.1  377.19
#Mann=8,-1,0
  4612.4   0.063       0  4679.3   0.035       0  4867.8    0.05       0
  4991.8    0.05       0  5004.5    0.05       0  5133.4   0.033       0
  6364.9   0.035       0  6462.7    0.05       0
Bank Sta=4991.8,5004.5
Exp/Cntr=0.3,0.1

Type RM Length L Ch R = 1,44981,466,466,466
BEGIN DESCRIPTION:
Prairie Creek44980.87
END DESCRIPTION:
XS GIS Cut Line= 3
      2705436.78      6828039.79      2705391.08      6828721.44
      2705347.02      6829690.26
#Sta/Elev= 30
  4326.8  377.59  4338.0  377.62  4388.1  372.06  4428.2  371.06  4501.9  371.70
  4562.7  371.72  4648.7  368.87  4849.2  367.44  4857.9  368.46  4863.0  364.14
  4869.2  367.70  4879.2  369.25  4903.3  363.24  4909.3  361.18  4949.4  370.40
  4979.5  371.01  4989.5  370.63  4999.5  365.51  5007.3  359.52  5023.2  359.43
  5023.7  358.93  5035.9  359.43  5039.6  363.55  5059.6  368.14  5069.6  368.57
  5319.9  367.74  5690.2  376.36  5750.3  375.74  5850.4  377.03  5979.8  374.97
#Mann=6,-1,0
  4326.8   0.094       0  4501.9   0.063       0  4562.7   0.094       0
  4903.3    0.05       0  5023.2    0.05       0  5035.9    0.05       0
Bank Sta=5023.2,5035.9
Exp/Cntr=0.3,0.1

Type RM Length L Ch R = 1,44515,400,400,400
BEGIN DESCRIPTION:
Prairie Creek44514.69
END DESCRIPTION:
XS GIS Cut Line= 3
      2704995.34      6828064.45      2704957.29      6828820.41
      2704810.74      6829579.07
#Sta/Elev= 30
  4252.5  375.58  4269.1  376.42  4289.1  375.72  4336.5  368.93  4359.2  369.95
  4383.4  368.86  4489.3  366.82  4519.4  367.44  4569.5  364.21  4579.5  364.38
  4609.5  367.79  4651.6  367.48  4848.6  367.60  4889.9  366.95  4929.9  364.80
  4949.9  367.21  4970.0  367.25  4980.0  365.64  4993.6  359.16  4994.1  358.66
  5006.4  359.16  5012.3  359.33  5030.4  365.54  5044.1  367.09  5142.4  366.86
  5213.7  370.39  5366.5  373.30  5682.2  375.69  5722.9  374.73  5782.1  375.32
#Mann=6,-1,0
  4252.5   0.063       0  4383.4   0.125       0  4651.6   0.063       0
  4848.6    0.05       0  4993.6    0.05       0  5006.4    0.05       0
Bank Sta=4993.6,5006.4
Exp/Cntr=0.3,0.1
