--- Prairie Creek Trib E.prj (project) ---

Proj Title=Prairie Creek Trib E Base Level Engineering
Current Plan=p01
Default Exp/Contr=0.3,0.1
English Units
Geom File=g01
Flow File=f01
Plan File=p01
Y Axis Title=Elevation
X Axis Title(PF)=Main Channel Distance
X Axis Title(XS)=Station
BEGIN DESCRIPTION:
Prairie Creek Trib E
END DESCRIPTION:
DSS Export Rating Curves= 0
DSS Export Rating Curve Sorted= 0
DSS Export Volume Flow Curves= 0
DXF OffsetX= 0
DXF OffsetY= 0
DXF ScaleX= 1
DXF ScaleY= 10

--- Prairie Creek Trib E.p01 (plan) ---

Plan Title=Multiple Run
Program Version=4.10
Short Identifier=Multiple
Geom File=g01
Flow File=f01
Subcritical Flow
K Sum by GR= 0
Std Step Tol= 0.01
Critical Tol= 0.01
Num of Std Step Trials= 20
Max Error Tol= 0.3
Flow Tol Ratio= 0.001
Split Flow NTrial= 30
Split Flow Tol= 0.02
Split Flow Ratio= 0.02
Log Output Level= 0
Friction Slope Method= 1
Unsteady Friction Slope Method= 2
Unsteady Bridges Friction Slope Method= 1
Parabolic Critical Depth
Global Vel Dist= 1 , 1 , 1
Global Log Level= 0
CheckData=True
Encroach Param=-1 ,0,0, 0
BEGIN DESCRIPTION:
Multiple Run
END DESCRIPTION:
Computation Interval=1HOUR
Output Interval=1HOUR
Run HTab= 0
Run UNet= 0
Run PostProcess= 0
Run WQNet= 0
UNET Theta= 1
UNET Theta Warmup= 1
UNET ZTol= 0.02
UNET ZSATol= 0.05
UNET MxIter= 20
UNET MaxInSteps= 0
UNET DtIC= 0
UNET DtMin= 0
UNET MaxCRTS= 20
UNET WFStab= 2
UNET SFStab= 1
UNET WFX= 1
UNET SFX= 1
UNET DSS MLevel= 4
UNET DZMax Abort= 100
UNET Convert EG Bridges= 0
UNET Use Existing IB Tables=-1
UNET Froude Reduction=False
UNET Froude Limit= 1
UNET Froude Power= 10
UNET Time Slicing=0,0, 5
UNET Junction Losses=0
Instantaneous Interval=1HOUR
Write IC File= 0
Write IC File at Sim End=0
Echo Input=False
Echo Parameters=False
Echo Output=False
Write Detailed= 0
WQ AD Non Conservative
WQ ULTIMATE=-1
WQ Max Comp Step=1HOUR
WQ Output Interval=15MIN
WQ Output Selected Increments= 0
WQ Output face flow=0
WQ Output face velocity=0
WQ Output face area=0
WQ Output face dispersion=0
WQ Output cell volume=0
WQ Output cell surface area=0
WQ Output cell continuity=0
WQ Output cumulative cell continuity=0
WQ Output face conc=0
WQ Output face dconc_dx=0
WQ Output face courant=0
WQ Output face peclet=0
WQ Output face adv mass=0
WQ Output face disp mass=0
WQ Output cell mass=0
WQ Output cell source sink temp=0
WQ Output cell source sink nsm=0
WQ Output MaxMinRange=-1
WQ Daily Max Min Mean=-1
WQ Daily Range=0
WQ Daily Time=0
WQ Create Restart=0
WQ Fixed Restart=0
WQ System Summary=0
WQ Use Fixed Temperature=0
Sorting and Armoring Iterations= 10
XS Update Threshold= 0.02
Hydraulics Update Threshold= 0.02
Energy Slope Method= 1
Volume Change Method= 0
XS Weighting Method= 0
Number of US Weighted Cross Sections= 1
Number of DS Weighted Cross Sections= 1
Upstream XS Weight=0.25
Main XS Weight=0.5
Downstream XS Weight=0.25
Number of DS XS's Weighted with US Boundary= 1
Upstream Boundary Weight= 1
Weight of XSs Associated with US Boundary= 0
Number of US XS's Weighted with DS Boundary= 1
Downstream Boundary Weight= 0.5
Weight of XSs Associated with DS Boundary= 0.5
Sediment Output Level= 4
Mass or Volume Output= 0
Output Increment Type= 1
Profile and TS Output Increment= 10
XS Output Flag= 0
XS Output Increment= 10
Disregard all LS=0
Disregard all Conn=0
Disregard all Breaches=0
Disregard all Pumps=0

--- Prairie Creek Trib E.f01 (steady flow) ---

Flow Title=Multiple
Number of Profiles=7
Profile Names=10-year,25-year,50-year,1pct_min,100-year,1pct_plu,500-year
River Rch & RM= Prairie Creek Tr,Reach-1,11233
     233     295     342     198     394     786     522
River Rch & RM= Prairie Creek Tr,Reach-1,9086
     529     701     838     497     992    1979    1388
River Rch & RM= Prairie Creek Tr,Reach-1,3582
     637     853    1027     614    1224    2443    1737
River Rch & RM= Prairie Creek Tr,Reach-1,2837
     679     910    1097     655    1306    2607    1853
Boundary for River Rch & Prof#=Prairie Creek Tr,Reach-1,1
Up Type=0
Dn Type=3
Dn Slope=0.005
Boundary for River Rch & Prof#=Prairie Creek Tr,Reach-1,2
Up Type=0
Dn Type=3
Dn Slope=0.005
Boundary for River Rch & Prof#=Prairie Creek Tr,Reach-1,3
Up Type=0
Dn Type=3
Dn Slope=0.005
Boundary for River Rch & Prof#=Prairie Creek Tr,Reach-1,4
Up Type=0
Dn Type=3
Dn Slope=0.005
Boundary for River Rch & Prof#=Prairie Creek Tr,Reach-1,5
Up Type=0
Dn Type=3
Dn Slope=0.005
Boundary for River Rch & Prof#=Prairie Creek Tr,Reach-1,6
Up Type=0
Dn Type=3
Dn Slope=0.005
Boundary for River Rch & Prof#=Prairie Creek Tr,Reach-1,7
Up Type=0
Dn Type=3
Dn Slope=0.005

--- Prairie Creek Trib E.g01 (geometry) ---

Geom Title=Existing Conditions

River Reach=Prairie Creek Tr,Reach-1
Reach XY= 30
      2706876.00      6817661.00      2706491.22      6817561.24
      2705936.71      6817760.28      2705524.45      6817514.75
      2705081.69      6817459.06      2704778.28      6817216.13
      2704665.95      6817249.89      2704083.48      6816567.06
      2704115.94      6816401.00      2703784.11      6816167.07
      2703720.47      6815858.58      2703433.68      6815617.52
      2703332.69      6815320.29      2703088.00      6815359.83
      2702983.02      6815170.01      2702831.56      6815208.74
      2702524.41      6815014.68      2702372.33      6815053.30
      2702274.58      6814914.04      2702131.63      6814959.25
      2701865.50      6814812.22      2701236.79      6814859.32
      2701170.64      6814612.95      2701029.64      6814703.83
      2700772.68      6814702.96      2700528.70      6814466.36
      2700311.87      6814447.64      2700209.53      6814144.27
      2699820.47      6813913.38      2698626.00      6813961.00

Type RM Length L Ch R = 1,11233,126,126,126
BEGIN DESCRIPTION:
Prairie Creek Trib E11233.452
END DESCRIPTION:
XS GIS Cut Line= 3
      2706827.75      6817378.24      2706820.28      6817661.04
      2706818.53      6817880.24
#Sta/Elev= 30
  4717.1  386.23  4769.9  385.84  4779.9  385.29  4799.9  384.86  4819.9  385.00
  4829.9  384.76  4839.9  385.03  4849.9  384.56  4857.9  383.17  4858.2  382.67
  4861.7  382.67  4861.9  383.17  4869.9  384.03  4879.9  384.08  4909.9  386.16
  4919.9  386.21  4949.9  385.98  4979.9  384.60  5010.0  385.33  5040.0  385.23
  5050.0  385.37  5060.0  384.29  5070.0  383.71  5090.0  384.94  5130.0  384.59
  5140.0  384.26  5180.0  383.84  5200.0  384.89  5217.1  387.17  5219.2  387.17
#Mann=3,-1,0
  4717.1    0.05       0  4857.9    0.05       0  4861.9    0.05       0
Bank Sta=4857.9,4861.9
Exp/Cntr=0.3,0.1

Type RM Length L Ch R = 1,11107,159,159,159
BEGIN DESCRIPTION:
Prairie Creek Trib E11107.41
END DESCRIPTION:
XS GIS Cut Line= 3
      2706705.62      6817351.13      2706694.20      6817662.50
      2706689.61      6817892.88
#Sta/Elev= 30
  4690.0  384.72  4709.9  384.62  4779.9  382.41  4789.9  382.14  4799.9  382.25
  4815.5  381.98  4820.5  381.61  4840.0  382.31  4850.0  382.44  4870.0  382.37
  4880.0  381.99  4910.0  382.74  4950.0  382.64  4960.1  382.88  4970.1  382.76
  5050.1  383.14  5060.1  382.57  5070.1  382.45  5090.1  383.13  5100.1  382.80
  5130.1  382.44  5163.7  381.47  5170.1  381.40  5180.1  381.73  5220.1  381.77
  5226.5  381.36  5226.8  380.86  5230.3  380.86  5230.5  381.36  5232.0  381.36
#Mann=3,-1,0
  4690.0    0.05       0  5226.5    0.05       0  5230.5    0.05       0
Bank Sta=5226.5,5230.5
Exp/Cntr=0.3,0.1

Type RM Length L Ch R = 1,10948,142,142,142
BEGIN DESCRIPTION:
Prairie Creek Trib E10947.98
END DESCRIPTION:
XS GIS Cut Line= 3
      2706575.27      6817362.08      2706571.83      6817564.90
      2706577.52      6817844.39
#Sta/Elev= 30
  4798.5  382.34  4807.4  382.66  4817.4  381.71  4827.4  381.25  4857.4  381.19
  4877.4  381.44  4887.4  380.84  4907.4  380.90  4917.4  380.61  4927.4  379.70
  4937.4  379.22  4945.4  379.22  4945.7  378.72  4949.2  378.72  4949.4  379.22
  4967.4  379.75  4977.4  380.58  4987.4  380.93  5001.3  380.86  5027.5  381.34
  5107.5  381.86  5137.5  381.89  5177.5  381.39  5207.5  379.36  5217.5  379.22
  5227.5  379.48  5237.5  379.23  5247.5  379.97  5257.5  379.57  5280.9  379.92
#Mann=3,-1,0
  4798.5    0.05       0  4945.4    0.05       0  4949.4    0.05       0
Bank Sta=4945.4,4949.4
Exp/Cntr=0.3,0.1

Type RM Length L Ch R = 1,10806,149,149,149
BEGIN DESCRIPTION:
Prairie Creek Trib E10806.16
END DESCRIPTION:
XS GIS Cut Line= 3
      2706439.39      6817425.52      2706442.07      6817598.31
      2706451.20      6817837.02
#Sta/Elev= 30
  4831.0  381.10  4836.5  380.77  4846.5  380.77  4886.5  379.50  4906.5  379.58
  4916.5  378.68  4926.5  378.81  4933.0  378.47  4938.0  378.69  4946.5  378.42
  4966.5  377.11  4976.5  376.81  4996.5  376.60  5016.5  376.70  5036.5  376.27
  5046.5  376.50  5074.6  376.01  5074.8  375.51  5078.3  375.51  5078.6  376.01
  5086.6  376.56  5116.6  376.73  5136.6  377.26  5146.6  377.92  5176.6  377.22
  5206.6  378.17  5216.7  377.82  5226.7  377.85  5234.5  378.13  5242.7  378.09
#Mann=3,-1,0
  4831.0    0.05       0  5074.6    0.05       0  5078.6    0.05       0
Bank Sta=5074.6,5078.6
Exp/Cntr=0.3,0.1

Type RM Length L Ch R = 1,10657,116,116,116
BEGIN DESCRIPTION:
Prairie Creek Trib E10657.16
END DESCRIPTION:
XS GIS Cut Line= 3
      2706319.83      6817449.59      2706318.61      6817664.92
      2706322.72      6817806.43
#Sta/Elev= 30
  4788.2  379.43  4799.6  379.34  4809.6  378.98  4829.6  378.79  4839.6  378.44
  4849.6  377.59  4859.6  377.37  4869.6  377.44  4909.6  376.53  4919.6  376.45
  4929.6  375.73  4939.6  375.21  4969.6  374.61  4979.6  374.73  4999.1  373.98
  5003.5  373.98  5009.6  374.48  5017.6  373.80  5017.9  373.30  5021.4  373.30
  5021.6  373.80  5029.6  374.55  5039.6  375.20  5059.6  375.17  5069.6  374.98
  5090.3  376.01  5099.7  375.92  5109.7  376.47  5119.7  376.68  5145.1  376.70
#Mann=3,-1,0
  4788.2    0.05       0  5017.6    0.05       0  5021.6    0.05       0
Bank Sta=5017.6,5021.6
Exp/Cntr=0.3,0.1

Type RM Length L Ch R = 1,10541,105,105,105
BEGIN DESCRIPTION:
Mapping XS 491a881a
END DESCRIPTION:
XS GIS Cut Line= 3
      2706202.37      6817525.46      2706202.24      6817660.50
      2706213.09      6818023.59
#Sta/Elev= 30
  4864.5  374.98  4870.0  375.71  4880.0  375.60  4890.0  375.29  4930.0  374.69
  4960.0  373.58  4990.0  372.97  4997.3  373.17  5020.1  373.24  5038.1  372.68
  5038.3  372.18  5041.8  372.18  5042.1  372.68  5050.1  374.23  5060.1  373.90
  5070.1  374.78  5080.1  374.22  5100.1  375.09  5110.1  374.14  5120.1  374.14
  5130.1  374.40  5150.1  374.34  5160.1  374.01  5171.0  373.13  5190.1  372.92
  5210.1  373.55  5240.2  373.96  5260.2  374.84  5294.0  375.54  5362.8  375.51
#Mann=4,-1,0
  4864.5    0.05       0  5038.1    0.05       0  5042.1    0.05       0
  5171.0   0.063       0
Bank Sta=5038.1,5042.1
Exp/Cntr=0.3,0.1

Type RM Length L Ch R = 1,10436,182,182,182
BEGIN DESCRIPTION:
Mapping XS 1bd2ae17
END DESCRIPTION:
XS GIS Cut Line= 3
      2706095.77      6817526.48      2706097.78      6817664.18
      2706093.04      6818066.34
#Sta/Elev= 30
  4865.6  374.34  4880.1  374.27  4900.1  373.82  4950.1  373.10  4960.1  372.55
  4970.1  371.74  4988.1  371.33  4988.4  370.83  4991.9  370.83  4992.1  371.33
  5010.1  371.47  5020.1  372.02  5040.1  372.18  5050.1  371.65  5060.1  372.02
  5070.1  371.76  5080.1  372.18  5120.1  371.67  5140.1  371.97  5154.7  371.76
  5160.1  371.65  5170.1  372.09  5220.1  372.85  5300.3  373.09  5310.2  372.90
  5340.2  372.80  5350.2  373.07  5380.2  373.23  5400.2  373.70  5405.5  374.41
#Mann=5,-1,0
  4865.6    0.05       0  4988.1    0.05       0  4992.1    0.05       0
  5154.7   0.063       0  5300.3    0.05       0
Bank Sta=4988.1,4992.1
Exp/Cntr=0.3,0.1

Type RM Length L Ch R = 1,10254,133,133,133
BEGIN DESCRIPTION:
Prairie Creek Trib E10254.19
END DESCRIPTION:
XS GIS Cut Line= 3
      2705960.37      6817363.12      2705953.06      6817765.58
      2705967.97      6818076.79
#Sta/Elev= 30
  4601.6  373.87  4679.5  372.92  4699.5  371.66  4729.5  371.74  4739.5  370.39
  4749.5  370.72  4769.5  372.15  4829.5  371.13  4849.5  369.90  4877.5  369.45
  4877.8  368.95  4881.3  368.95  4881.5  369.45  4909.5  370.45  4919.5  369.90
  4959.5  370.82  4979.5  369.73  5019.6  369.98  5029.6  370.63  5039.6  370.16
  5079.6  370.82  5099.7  370.69  5109.7  371.27  5119.7  370.83  5139.7  370.75
  5219.8  371.39  5249.8  372.05  5269.9  371.68  5279.9  372.07  5315.7  372.15
#Mann=3,-1,0
  4601.6    0.05       0  4877.5    0.05       0  4881.5    0.05       0
Bank Sta=4877.5,4881.5
Exp/Cntr=0.3,0.1

Type RM Length L Ch R = 1,10121,84,84,84
BEGIN DESCRIPTION:
Mapping XS a2d3ad5f
END DESCRIPTION:
XS GIS Cut Line= 4
      2705902.37      6817235.95      2705833.97      6817730.25
      2705851.53      6818443.80      2705886.58      6818615.99
#Sta/Elev= 30
  4520.5  375.26  4535.7  375.60  4545.8  374.32  4607.4  373.32  4666.9  373.18
  4679.2  371.84  4717.4  371.46  4751.1  370.19  4757.8  370.80  4788.1  369.28
  4798.2  369.14  4808.3  370.17  4817.8  370.18  4899.7  369.01  4998.0  368.48
  4998.3  367.98  5001.8  367.98  5002.0  368.48  5520.4  372.04  5550.4  371.51
  5610.4  372.65  5620.4  373.70  5650.4  373.06  5690.5  374.49  5708.6  373.90
  5771.2  375.01  5829.1  376.42  5834.2  377.55  5842.7  377.88  5909.0  379.47
#Mann=3,-1,0
  4520.5    0.05       0  4998.0    0.05       0  5002.0    0.05       0
Bank Sta=4998,5002
Exp/Cntr=0.3,0.1

Type RM Length L Ch R = 1,10037,115,115,115
BEGIN DESCRIPTION:
Mapping XS db925d32
END DESCRIPTION:
XS GIS Cut Line= 3
      2705801.30      6817224.44      2705742.83      6817853.67
      2705826.23      6818642.13
#Sta/Elev= 30
  4529.3  374.18  4576.1  373.22  4596.1  373.60  4616.2  372.14  4641.0  371.45
  4656.4  370.35  4726.7  369.79  4756.8  368.69  4797.0  368.99  4807.1  367.86
  4837.2  369.14  4859.5  369.24  4887.4  367.51  4987.8  366.83  4997.9  367.44
  4998.0  366.83  4998.3  366.33  5001.8  366.33  5002.0  366.83  5007.9  367.61
  5018.0  367.28  5118.4  369.05  5329.2  369.62  5651.3  372.45  5715.5  373.36
  5751.8  375.21  5822.2  375.02  5882.6  376.31  5912.7  378.51  5954.1  378.33
#Mann=3,-1,0
  4529.3    0.05       0  4998.0    0.05       0  5002.0    0.05       0
Bank Sta=4998,5002
Exp/Cntr=0.3,0.1

Type RM Length L Ch R = 1,9922,132,132,132
BEGIN DESCRIPTION:
Mapping XS 48f5faa3
END DESCRIPTION:
XS GIS Cut Line= 4
      2705731.11      6817225.95      2705659.84      6817732.41
      2705630.54      6818221.47      2705800.27      6818641.60
#Sta/Elev= 30
  4610.6  373.39  4635.9  373.42  4646.0  372.19  4666.2  371.41  4726.8  370.59
  4797.5  368.28  4868.2  368.02  4895.9  366.93  4998.0  365.74  4998.3  365.24
  5001.8  365.24  5002.0  365.74  5009.5  366.38  5049.9  365.93  5070.1  366.88
  5114.7  367.04  5200.8  368.79  5391.1  369.19  5511.3  371.54  5644.6  372.95
  5717.0  372.20  5730.1  372.64  5740.9  371.88  5746.5  372.59  5829.7  373.40
  5891.9  375.53  5978.2  375.65  6014.8  376.89  6032.1  378.42  6065.1  378.22
#Mann=3,-1,0
  4610.6    0.05       0  4998.0    0.05       0  5002.0    0.05       0
Bank Sta=4998,5002
Exp/Cntr=0.3,0.1

Type RM Length L Ch R = 1,9790,117,117,117
BEGIN DESCRIPTION:
Mapping XS a7b6592a
END DESCRIPTION:
XS GIS Cut Line= 4
      2705629.83      6817223.63      2705547.66      6817638.04
      2705557.94      6818100.45      2705791.59      6818652.22
#Sta/Elev= 30
  4668.4  371.64  4706.5  371.10  4726.9  369.68  4769.0  368.46  4820.2  367.58
  4849.2  367.82  4871.4  366.46  4941.0  366.60  4951.2  365.65  4961.4  365.86
  4998.0  364.37  4998.3  363.87  5001.8  363.87  5002.0  364.37  5089.8  366.36
  5123.8  366.47  5173.9  368.05  5323.9  368.22  5589.4  372.73  5771.5  372.59
  5789.8  371.93  5803.8  372.48  5813.4  371.69  5825.5  372.70  5866.2  372.66
  5966.4  375.41  6064.4  375.85  6095.7  376.87  6124.8  378.75  6152.6  378.46
#Mann=3,-1,0
  4668.4    0.05       0  4998.0    0.05       0  5002.0    0.05       0
Bank Sta=4998,5002
Exp/Cntr=0.3,0.1

Type RM Length L Ch R = 1,9673,149,149,149
BEGIN DESCRIPTION:
Mapping XS 64b0dd31
END DESCRIPTION:
XS GIS Cut Line= 3
      2705525.74      6817230.47      2705421.90      6817684.15
      2705115.48      6818592.33
#Sta/Elev= 30
  4712.5  368.87  4754.1  367.76  4774.0  368.08  4784.9  366.99  4938.7  365.85
  4956.0  364.88  4961.1  365.59  4969.5  364.52  4979.8  365.89  4998.0  362.87
  4998.3  362.37  5001.8  362.37  5002.0  362.87  5004.0  364.18  5020.8  362.87
  5061.8  364.68  5154.2  367.19  5458.3  367.01  5565.1  366.12  5773.0  367.24
  5841.2  366.79  5898.9  367.81  5945.0  367.09  5961.8  367.96  5967.1  367.13
  6018.9  369.08  6030.0  368.54  6082.2  369.24  6113.9  370.76  6136.4  370.30
#Mann=3,-1,0
  4712.5    0.05       0  4998.0    0.05       0  5002.0    0.05       0
Bank Sta=4998,5002
Exp/Cntr=0.3,0.1

Type RM Length L Ch R = 1,9524,156,156,156
BEGIN DESCRIPTION:
Mapping XS 2f0bad9f
END DESCRIPTION:
XS GIS Cut Line= 3
      2705419.14      6817234.15      2705162.61      6817889.45
      2704906.49      6818413.16
#Sta/Elev= 30
  4715.2  366.78  4808.5  365.85  4829.9  366.37  4876.5  363.94  4930.8  362.83
  4955.2  364.23  4969.2  363.82  4998.0  362.53  4998.3  362.03  5002.0  362.53
  5007.8  362.59  5033.9  364.05  5069.1  364.28  5087.7  363.61  5118.1  364.57
  5179.4  364.63  5238.0  364.48  5302.5  365.59  5345.9  364.89  5441.3  365.20
  5463.9  364.53  5514.4  364.57  5531.4  365.63  5537.0  364.76  5581.6  364.90
  5784.6  367.45  5852.1  369.26  5919.7  368.81  5970.3  370.44  6001.9  370.27
#Mann=7,-1,0
  4715.2    0.05       0  4969.2    0.07       0  4998.0    0.07       0
  5002.0    0.07       0  5007.8    0.05       0  5179.4    0.07       0
  5581.6    0.05       0
Bank Sta=4998,5002
Exp/Cntr=0.3,0.1

Type RM Length L Ch R = 1,9368,282,282,282
BEGIN DESCRIPTION:
Mapping XS 799093d0
END DESCRIPTION:
XS GIS Cut Line= 3
      2705292.02      6817225.15      2705145.54      6817497.29
      2704708.17      6818236.66
#Sta/Elev= 30
  4776.0  366.12  4850.8  363.61  4903.3  363.33  4909.0  362.68  4953.0  361.88
  4985.3  362.31  4998.0  361.82  4998.3  361.32  5001.8  361.32  5002.0  361.82
  5051.0  362.68  5066.6  361.82  5084.3  362.53  5124.2  362.77  5137.5  363.78
  5159.1  363.90  5174.5  363.20  5196.5  363.67  5240.4  362.82  5248.7  362.11
  5295.2  363.40  5334.4  364.06  5504.1  364.49  5605.5  363.85  5685.5  365.62
  5774.9  366.75  5796.7  368.00  5861.0  368.05  5913.7  369.94  5944.1  369.50
#Mann=5,-1,0
  4776.0    0.05       0  4998.0    0.05       0  5002.0    0.05       0
  5196.5    0.07       0  5295.2    0.05       0
Bank Sta=4998,5002
Exp/Cntr=0.3,0.1

Type RM Length L Ch R = 1,9086,218,218,218
BEGIN DESCRIPTION:
Prairie Creek Trib E9085.58
END DESCRIPTION:
XS GIS Cut Line= 3
      2705247.35      6817217.19      2704966.23      6817363.18
      2704541.03      6817443.58
#Sta/Elev= 30
  4688.6  366.37  4707.4  366.25  4713.0  365.19  4729.5  364.61  4825.3  363.96
  4840.1  363.07  4906.4  361.77  4960.6  361.41  4972.8  360.59  4989.3  360.71
  5002.7  359.33  5015.6  359.40  5036.1  361.18  5060.4  361.50  5066.7  362.10
  5125.4  361.64  5135.9  358.77  5136.2  358.27  5139.9  358.77  5148.1  360.73
  5158.3  361.53  5168.4  360.70  5182.9  362.01  5199.0  361.05  5219.3  361.70
  5242.7  360.84  5287.6  360.43  5331.3  361.64  5351.6  363.48  5438.1  364.60
#Mann=5,-1,0
  4688.6    0.05       0  5060.4    0.16       0  5135.9    0.05       0
  5139.9    0.16       0  5242.7    0.05       0
Bank Sta=5135.9,5139.9
Exp/Cntr=0.3,0.1

Type RM Length L Ch R = 1,8868,309,309,309
BEGIN DESCRIPTION:
Prairie Creek Trib E8868.29
END DESCRIPTION:
XS GIS Cut Line= 3
      2705062.60      6817069.22      2704800.01      6817238.18
      2704540.79      6817401.82
#Sta/Elev= 30
  4690.5  365.74  4718.8  364.53  4761.1  364.05  4776.3  362.70  4921.6  360.86
  4948.6  359.87  4963.8  360.10  4971.8  360.87  4994.2  360.54  5002.2  359.88
  5017.2  360.15  5021.3  359.87  5036.6  360.55  5066.6  359.87  5079.0  360.85
  5094.3  359.97  5130.7  361.05  5146.0  359.43  5151.9  360.47  5169.1  360.32
  5201.7  358.88  5201.9  358.38  5205.4  358.38  5205.7  358.88  5219.0  359.24
  5224.0  360.21  5232.2  360.58  5246.1  362.29  5285.1  363.56  5309.3  363.76
#Mann=7,-1,0
  4690.5    0.05       0  5017.2    0.16       0  5169.1    0.05       0
  5201.7    0.05       0  5205.7    0.05       0  5224.0    0.07       0
  5285.1    0.05       0
Bank Sta=5201.7,5205.7
Exp/Cntr=0.3,0.1

Type RM Length L Ch R = 1,8559,249,249,249
BEGIN DESCRIPTION:
Prairie Creek Trib E8559.02
END DESCRIPTION:
XS GIS Cut Line= 3
      2704860.38      6816970.77      2704558.68      6817145.77
      2704405.94      6817269.58
#Sta/Elev= 30
  4652.7  362.25  4679.1  362.06  4706.4  360.97  4737.9  360.97  4773.4  360.40
  4808.2  359.14  4845.5  359.28  4854.3  358.13  4867.0  358.95  4906.7  358.75
  4920.0  357.97  4925.8  358.70  4941.6  359.05  4947.3  359.70  4951.5  359.44
  4957.3  359.09  4978.8  359.22  4984.6  359.77  4991.0  357.83  4991.3  357.33
  4994.8  357.33  4995.0  357.83  5000.1  358.01  5006.6  359.04  5017.4  358.97
  5043.3  358.58  5070.5  359.67  5084.9  361.18  5134.2  362.19  5198.1  363.39
#Mann=7,-1,0
  4652.7    0.05       0  4906.7    0.12       0  4951.5    0.16       0
  4991.0    0.07       0  4995.0    0.16       0  5017.4    0.07       0
  5134.2    0.05       0
Bank Sta=4991,4995
Exp/Cntr=0.3,0.1

Type RM Length L Ch R = 1,8310,228,228,228
BEGIN DESCRIPTION:
Prairie Creek Trib E8310.1
END DESCRIPTION:
XS GIS Cut Line= 3
      2704744.05      6816896.71      2704391.53      6816980.93
      2704175.50      6817025.38
#Sta/Elev= 30
  4640.5  360.89  4682.6  360.25  4689.9  360.54  4761.6  359.01  4766.8  358.58
  4787.1  358.87  4803.0  358.30  4814.0  357.28  4844.1  358.42  4893.0  357.92
  4898.2  358.59  4905.8  358.37  4916.1  357.69  4924.4  352.97  4924.6  352.47
  4928.1  352.47  4928.4  352.97  4935.1  357.93  4940.3  357.72  4946.6  358.33
  4957.2  357.83  4977.2  357.71  4988.1  357.08  5002.9  357.10  5018.8  357.51
  5031.1  359.24  5093.4  360.40  5161.7  361.50  5182.1  362.29  5223.5  363.02
#Mann=6,-1,0
  4640.5    0.05       0  4787.1    0.12       0  4924.4    0.07       0
  4928.4    0.12       0  4946.6    0.07       0  5093.4    0.05       0
Bank Sta=4924.4,4928.4
Exp/Cntr=0.3,0.1

Type RM Length L Ch R = 1,8082,168,168,168
BEGIN DESCRIPTION:
Prairie Creek Trib E8081.56
END DESCRIPTION:
XS GIS Cut Line= 3
      2704798.05      6816798.49      2704301.03      6816785.92
      2703699.57      6816777.46
#Sta/Elev= 30
  4502.8  363.03  4600.6  361.48  4605.6  361.78  4674.9  360.80  4764.9  358.10
  4789.0  358.24  4865.0  356.70  4895.0  356.65  4915.0  354.61  4925.0  355.20
  4935.0  356.83  4945.0  355.79  4963.0  352.19  4963.3  351.69  4966.8  351.69
  4967.0  352.19  4975.0  354.86  4985.0  355.37  4998.3  355.82  5042.7  355.96
  5055.0  356.53  5065.0  357.71  5075.0  357.30  5085.9  357.69  5295.0  358.47
  5395.1  358.16  5405.1  357.65  5425.1  358.43  5525.1  359.44  5601.5  361.22
#Mann=6,-1,0
  4502.8    0.05       0  4789.0    0.12       0  4963.0    0.07       0
  4967.0    0.12       0  5042.7    0.07       0  5085.9    0.05       0
Bank Sta=4963,4967
Exp/Cntr=0.3,0.1

Type RM Length L Ch R = 1,7914,368,368,368
BEGIN DESCRIPTION:
Prairie Creek Trib E7914.02
END DESCRIPTION:
XS GIS Cut Line= 3
      2704717.24      6816662.88      2704179.13      6816667.56
      2703644.47      6816664.53
#Sta/Elev= 30
  4465.2  364.71  4536.4  363.26  4546.4  363.81  4566.4  361.92  4606.4  360.35
  4676.5  359.15  4726.5  357.61  4836.5  355.81  4856.5  355.93  4866.5  356.61
  4876.5  355.13  4884.5  351.71  4884.7  351.21  4888.2  351.21  4888.5  351.71
  4896.5  354.35  4906.5  355.69  4951.3  356.06  4976.5  354.79  4986.5  355.25
  4996.5  354.36  5002.4  353.19  5007.4  353.19  5016.5  354.75  5046.5  355.81
  5114.1  355.76  5274.7  356.24  5296.5  355.78  5496.5  360.69  5538.0  360.68
#Mann=5,-1,0
  4465.2    0.05       0  4884.5    0.07       0  4888.5    0.05       0
  4951.3    0.07       0  5114.1    0.05       0
Bank Sta=4884.5,4888.5
Exp/Cntr=0.3,0.1

Type RM Length L Ch R = 1,7546,355,355,355
BEGIN DESCRIPTION:
Prairie Creek Trib E7546.07
END DESCRIPTION:
XS GIS Cut Line= 3
      2704475.55      6816333.99      2704083.26      6816373.15
      2703522.75      6816416.13
#Sta/Elev= 30
  4610.0  368.39  4649.7  367.15  4669.8  365.62  4733.0  362.78  4780.4  359.23
  4810.5  358.10  4850.7  355.80  4911.0  355.09  4929.2  355.30  4941.2  354.32
  4961.3  353.49  5004.2  353.55  5039.1  354.79  5044.1  354.49  5049.6  351.68
  5049.9  351.18  5053.4  351.18  5053.6  351.68  5061.7  354.59  5081.7  354.24
  5091.8  353.52  5131.9  354.26  5232.2  353.77  5242.2  353.39  5300.3  353.85
  5402.7  356.59  5430.8  356.69  5492.9  358.21  5533.0  359.82  5566.4  360.61
#Mann=3,-1,0
  4610.0    0.05       0  5049.6    0.05       0  5053.6    0.05       0
Bank Sta=5049.6,5053.6
Exp/Cntr=0.3,0.1

Type RM Length L Ch R = 1,7191,233,233,233
BEGIN DESCRIPTION:
Prairie Creek Trib E7191.04
END DESCRIPTION:
XS GIS Cut Line= 3
      2704224.32      6816160.55      2703798.10      6816185.96
      2703521.62      6816221.26
#Sta/Elev= 30
  4575.2  359.04  4613.6  356.59  4633.6  356.16  4643.6  355.42  4673.7  354.40
  4773.9  353.65  4793.9  354.00  4824.0  353.03  4831.9  352.40  4836.9  353.43
  4844.0  351.26  4854.0  354.08  4864.0  354.19  4874.1  353.45  4894.1  352.68
  4934.2  353.07  4964.2  352.83  5005.9  351.95  5022.5  351.14  5022.7  350.64
  5026.2  350.64  5026.5  351.14  5034.5  352.11  5044.6  352.59  5115.2  354.03
  5125.3  353.85  5195.8  356.58  5240.3  357.78  5256.3  358.78  5280.9  359.51
#Mann=3,-1,0
  4575.2    0.05       0  5022.5    0.05       0  5026.5    0.05       0
Bank Sta=5022.5,5026.5
Exp/Cntr=0.3,0.1

Type RM Length L Ch R = 1,6958,96,96,96
BEGIN DESCRIPTION:
Prairie Creek Trib E6958.23
END DESCRIPTION:
XS GIS Cut Line= 3
      2704219.93      6816013.69      2703752.92      6815990.12
      2703500.14      6815988.27
#Sta/Elev= 30
  4534.7  357.91  4598.7  356.11  4618.7  355.97  4638.8  355.50  4668.8  355.41
  4685.5  355.11  4698.8  355.26  4809.0  353.80  4829.0  353.81  4889.8  352.97
  4909.1  352.49  4929.1  352.63  4949.2  351.92  4979.2  352.83  4987.2  349.51
  4987.5  349.01  4991.0  349.01  4991.2  349.51  4998.3  352.53  5002.3  352.53
  5009.2  352.97  5019.2  352.16  5029.2  351.88  5039.2  352.37  5049.2  351.82
  5079.2  352.95  5099.2  353.15  5129.2  354.01  5169.2  355.94  5255.1  357.77
#Mann=3,-1,0
  4534.7    0.05       0  4987.2    0.05       0  4991.2    0.05       0
Bank Sta=4987.2,4991.2
Exp/Cntr=0.3,0.1

Type RM Length L Ch R = 1,6862,143,143,143
BEGIN DESCRIPTION:
Prairie Creek Trib E6862.1
END DESCRIPTION:
XS GIS Cut Line= 3
      2704146.36      6815901.62      2703724.01      6815903.74
      2703489.13      6815890.68
#Sta/Elev= 30
  4579.8  357.18  4600.2  356.89  4610.2  356.45  4630.2  356.39  4680.2  355.55
  4690.2  355.61  4760.2  354.36  4800.2  354.12  4840.2  353.32  4930.2  352.94
  4940.2  353.22  4950.2  352.76  4960.2  353.22  4980.2  351.44  4988.2  350.05
  4988.4  349.55  4991.9  349.55  4992.2  350.05  4998.7  352.08  5030.2  352.13
  5040.2  351.74  5060.3  351.40  5070.3  351.51  5110.3  353.11  5138.5  354.66
  5143.5  354.37  5160.4  355.19  5210.5  356.50  5230.5  357.32  5237.4  357.22
#Mann=3,-1,0
  4579.8    0.05       0  4988.2    0.05       0  4992.2    0.05       0
Bank Sta=4988.2,4992.2
Exp/Cntr=0.3,0.1

Type RM Length L Ch R = 1,6719,130,130,130
BEGIN DESCRIPTION:
Prairie Creek Trib E6719.45
END DESCRIPTION:
XS GIS Cut Line= 3
      2703988.53      6815679.39      2703653.25      6815789.14
      2703510.93      6815826.00
#Sta/Elev= 30
  4647.6  353.13  4681.8  353.55  4723.9  353.44  4863.8  352.48  4871.2  352.04
  4890.4  352.43  4895.7  351.96  4913.3  353.21  4927.6  352.03  4934.4  349.43
  4944.9  348.50  4954.1  349.21  4959.4  350.99  4965.9  349.40  4974.4  348.25
  4974.7  347.75  4978.2  347.75  4978.4  348.25  4986.0  349.24  4991.3  349.43
  4996.3  350.83  5025.6  351.46  5059.5  351.02  5066.2  351.80  5071.3  351.84
  5080.2  352.33  5100.8  352.41  5111.9  353.23  5131.8  353.72  5147.4  354.74
#Mann=3,-1,0
  4647.6    0.05       0  4974.4    0.05       0  4978.4    0.05       0
Bank Sta=4974.4,4978.4
Exp/Cntr=0.3,0.1

Type RM Length L Ch R = 1,6589,122,122,122
BEGIN DESCRIPTION:
Prairie Creek Trib E6588.95
END DESCRIPTION:
XS GIS Cut Line= 3
      2703861.64      6815309.42      2703592.31      6815680.60
      2703450.84      6815855.82
#Sta/Elev= 30
  4544.4  354.33  4657.5  353.85  4699.8  352.44  4821.1  352.23  4835.8  351.65
  4842.9  349.96  4850.5  349.61  4856.7  349.67  4865.2  352.18  4871.4  350.72
  4900.8  351.33  4906.9  349.84  4915.5  351.50  4921.6  349.21  4929.4  350.72
  4936.3  350.17  4940.5  348.43  4940.8  347.93  4944.3  347.93  4944.5  348.43
  4951.0  348.44  4965.7  351.03  4978.8  352.03  4992.8  351.02  5003.0  351.04
  5015.5  349.43  5065.1  351.33  5135.4  352.97  5178.6  355.37  5228.2  357.10
#Mann=3,-1,0
  4544.4    0.05       0  4940.5    0.05       0  4944.5    0.05       0
Bank Sta=4940.5,4944.5
Exp/Cntr=0.3,0.1

Type RM Length L Ch R = 1,6467,289,289,289
BEGIN DESCRIPTION:
Prairie Creek Trib E6467.49
END DESCRIPTION:
XS GIS Cut Line= 3
      2703689.81      6815108.04      2703477.01      6815659.59
      2703418.02      6815837.81
#Sta/Elev= 30
  4410.9  354.14  4424.8  354.13  4438.1  353.44  4547.3  352.62  4601.9  352.91
  4607.2  352.13  4656.4  352.29  4692.8  351.29  4765.6  350.75  4789.2  349.56
  4820.2  350.26  4896.4  349.87  4917.8  350.40  4940.0  349.92  4971.4  350.33
  4982.2  349.24  4989.3  347.24  4994.6  347.62  4998.2  346.27  4998.4  345.77
  5001.9  345.77  5002.2  346.27  5005.5  346.27  5014.1  349.00  5020.3  349.45
  5025.5  351.07  5035.2  351.74  5045.7  351.28  5066.8  352.88  5189.8  356.91
#Mann=3,-1,0
  4410.9    0.05       0  4998.2    0.05       0  5002.2    0.05       0
Bank Sta=4998.2,5002.2
Exp/Cntr=0.3,0.1

Type RM Length L Ch R = 1,6178,172,172,172
BEGIN DESCRIPTION:
Prairie Creek Trib E6177.13
END DESCRIPTION:
XS GIS Cut Line= 3
      2703492.27      6814871.59      2703408.74      6815397.92
      2703353.75      6815796.32
#Sta/Elev= 30
  4471.1  359.11  4511.0  356.45  4612.3  351.95  4632.5  351.55  4713.5  351.84
  4731.6  351.25  4764.1  351.70  4905.9  350.49  4916.0  349.51  4923.4  345.21
  4936.3  346.27  4954.5  342.79  4954.8  342.29  4958.3  342.29  4958.5  342.79
  4966.6  346.89  4976.8  349.06  4979.9  349.03  5014.3  348.89  5027.3  349.29
  5047.5  348.79  5056.6  349.36  5061.6  348.83  5067.7  349.69  5077.8  349.77
  5098.0  349.28  5188.8  349.79  5340.3  353.74  5400.8  355.02  5406.2  354.70
#Mann=5,-1,0
  4471.1    0.05       0  4954.5    0.07       0  4958.5    0.05       0
  4979.9    0.16       0  5014.3    0.05       0
Bank Sta=4954.5,4958.5
Exp/Cntr=0.3,0.1

Type RM Length L Ch R = 1,6006,94,94,94
BEGIN DESCRIPTION:
Prairie Creek Trib E5992.93
END DESCRIPTION:
XS GIS Cut Line= 3
      2703288.44      6814783.78      2703279.41      6815352.61
      2703282.19      6815967.10
#Sta/Elev= 30
  4431.1  358.17  4438.3  358.39  4458.3  357.53  4498.3  355.05  4598.3  353.01
  4628.3  353.00  4698.4  350.93  4748.4  351.01  4798.4  350.01  4808.4  349.35
  4858.4  349.43  4888.4  348.14  4896.6  348.82  4918.4  348.55  4928.4  347.78
  4936.4  344.15  4936.6  343.65  4940.1  343.65  4940.4  344.15  4948.4  345.12
  4958.4  348.06  4989.8  347.93  5018.4  347.56  5058.4  348.69  5116.1  348.90
  5318.4  350.83  5488.4  353.22  5568.4  355.26  5578.4  356.13  5614.5  357.14
#Mann=5,-1,0
  4431.1    0.05       0  4936.4    0.07       0  4940.4    0.05       0
  4989.8    0.16       0  5116.1    0.05       0
Bank Sta=4936.4,4940.4
Exp/Cntr=0.3,0.1

Type RM Length L Ch R = 1,5912,355,355,355
BEGIN DESCRIPTION:
Prairie Creek Trib E5911.86
END DESCRIPTION:
XS GIS Cut Line= 3
      2703212.97      6814740.57      2703199.84      6815311.34
      2703190.54      6815990.36
#Sta/Elev= 30
  4429.7  358.39  4610.2  351.68  4630.2  352.09  4730.2  350.13  4800.2  349.78
  4890.3  347.58  4952.7  347.64  4970.3  348.12  4980.3  347.82  4990.3  348.40
  4995.9  342.11  4996.2  341.61  4999.7  341.61  4999.9  342.11  5002.9  342.11
  5004.4  343.06  5010.3  346.82  5013.8  347.22  5020.3  347.97  5050.3  347.37
  5080.3  347.96  5150.3  347.87  5210.3  349.11  5250.3  349.07  5380.3  350.46
  5470.3  351.76  5560.3  353.79  5570.3  353.66  5600.3  355.46  5679.7  356.75
#Mann=5,-1,0
  4429.7    0.05       0  4995.9    0.05       0  4999.9    0.05       0
  5004.4    0.16       0  5013.8    0.05       0
Bank Sta=4995.9,4999.9
Exp/Cntr=0.3,0.1

Type RM Length L Ch R = 1,5557,147,147,147
BEGIN DESCRIPTION:
Prairie Creek Trib E5556.6
END DESCRIPTION:
XS GIS Cut Line= 3
      2702991.99      6814957.94      2702982.72      6815172.45
      2702974.60      6815596.26
#Sta/Elev= 30
  4787.8  348.86  4840.9  347.80  4881.0  347.49  4891.0  347.00  4901.0  347.39
  4921.0  346.95  4931.0  347.26  4951.0  346.43  4970.4  346.40  5002.5  346.63
  5021.1  346.16  5031.1  346.72  5041.1  345.31  5049.1  340.78  5049.3  340.28
  5052.8  340.28  5053.1  340.78  5061.1  344.97  5071.1  346.40  5094.3  347.08
  5149.3  346.62  5161.1  346.72  5191.1  345.61  5221.1  346.02  5291.1  348.17
  5311.1  348.40  5321.1  349.09  5351.1  349.50  5391.1  350.93  5426.4  351.23
#Mann=5,-1,0
  4787.8    0.05       0  4970.4    0.16       0  5049.1    0.07       0
  5053.1    0.16       0  5149.3   0.035       0
Bank Sta=5049.1,5053.1
Exp/Cntr=0.3,0.1

Type RM Length L Ch R = 1,5410,146,146,146
BEGIN DESCRIPTION:
Prairie Creek Trib E5409.93
END DESCRIPTION:
XS GIS Cut Line= 3
      2702883.67      6814877.79      2702850.31      6815214.77
      2702821.95      6815493.40
#Sta/Elev= 30
  4664.8  348.95  4828.8  345.85  4859.0  345.65  4879.1  346.27  4889.1  346.22
  4909.2  345.30  4919.3  345.74  4929.3  345.15  4949.4  345.71  4959.4  345.31
  4983.8  345.82  4995.5  345.27  5009.7  345.90  5049.9  345.87  5060.0  346.31
  5070.0  343.95  5078.1  339.65  5078.3  339.15  5081.8  339.15  5082.1  339.65
  5090.1  342.13  5095.2  342.09  5099.1  345.20  5100.3  346.16  5120.3  345.55
  5150.4  345.21  5160.5  345.74  5220.8  346.87  5250.9  348.48  5283.5  349.62
#Mann=5,-1,0
  4664.8    0.05       0  4983.8    0.16       0  5078.1    0.07       0
  5082.1    0.16       0  5099.1    0.05       0
Bank Sta=5078.1,5082.1
Exp/Cntr=0.3,0.1

Type RM Length L Ch R = 1,5264,252,252,252
BEGIN DESCRIPTION:
Prairie Creek Trib E5264.23
END DESCRIPTION:
XS GIS Cut Line= 3
      2702761.63      6814829.61      2702721.03      6815162.05
      2702675.43      6815552.79
#Sta/Elev= 30
  4673.1  347.99  4678.9  347.57  4734.9  347.07  4795.4  345.47  4835.7  345.16
  4855.8  344.55  4928.6  344.04  4966.7  344.93  4986.8  344.56  4996.9  343.71
  5010.1  345.29  5047.2  345.03  5060.5  345.48  5067.4  345.88  5077.4  342.10
  5093.5  341.48  5098.6  338.56  5105.6  338.29  5105.9  337.79  5109.4  337.79
  5109.6  338.29  5117.7  342.11  5127.8  345.63  5141.7  345.84  5158.0  345.31
  5208.3  346.28  5228.4  346.22  5265.4  348.21  5329.1  349.11  5401.4  351.62
#Mann=5,-1,0
  4673.1    0.05       0  5060.5    0.16       0  5105.6    0.05       0
  5109.6    0.16       0  5141.7    0.05       0
Bank Sta=5105.6,5109.6
Exp/Cntr=0.3,0.1

Type RM Length L Ch R = 1,5012,180,180,180
BEGIN DESCRIPTION:
Prairie Creek Trib E5011.72
END DESCRIPTION:
XS GIS Cut Line= 3
      2702547.14      6814725.15      2702520.33      6815016.81
      2702495.97      6815362.57
#Sta/Elev= 30
  4710.6  347.77  4716.5  347.19  4788.8  345.57  4806.9  345.58  4826.9  344.93
  4987.6  343.10  4994.4  342.36  5003.1  342.85  5017.7  342.48  5057.8  343.27
  5077.9  343.80  5087.9  344.49  5096.6  343.82  5097.9  343.72  5105.9  338.34
  5106.2  337.84  5109.7  337.84  5109.9  338.34  5118.0  344.33  5134.6  344.21
  5139.6  342.21  5148.0  344.24  5158.1  343.37  5178.1  343.71  5188.1  344.41
  5238.3  344.22  5259.3  345.59  5268.3  346.10  5280.9  345.38  5350.1  347.21
#Mann=6,-1,0
  4710.6   0.035       0  4788.8    0.05       0  5096.6    0.16       0
  5105.9    0.05       0  5109.9    0.16       0  5259.3    0.05       0
Bank Sta=5105.9,5109.9
Exp/Cntr=0.3,0.1

Type RM Length L Ch R = 1,4832,309,309,309
BEGIN DESCRIPTION:
Prairie Creek Trib E4832.05
END DESCRIPTION:
XS GIS Cut Line= 3
      2702380.80      6814745.19      2702357.71      6815051.23
      2702330.01      6815365.81
#Sta/Elev= 30
  4700.1  347.48  4736.0  345.72  4786.1  343.93  4856.3  342.92  4926.5  342.63
  4946.6  341.56  4956.6  340.52  4962.4  339.70  4967.5  338.25  4974.7  337.34
  4974.9  336.84  4978.4  336.84  4978.7  337.34  4985.2  337.88  4996.7  340.39
  5004.4  341.56  5009.4  341.56  5016.8  342.48  5026.9  342.92  5067.0  343.49
  5077.0  343.00  5117.2  343.59  5137.3  343.15  5192.8  344.38  5200.0  344.08
  5247.7  344.57  5277.8  345.44  5307.2  347.02  5312.2  346.37  5322.8  346.66
#Mann=5,-1,0
  4700.1    0.05       0  4974.7    0.07       0  4978.7    0.05       0
  4985.2    0.16       0  5192.8    0.05       0
Bank Sta=4974.7,4978.7
Exp/Cntr=0.3,0.1

Type RM Length L Ch R = 1,4523,236,236,236
BEGIN DESCRIPTION:
Prairie Creek Trib E4522.75
END DESCRIPTION:
XS GIS Cut Line= 3
      2702183.25      6814704.43      2702143.54      6814964.99
      2702106.84      6815357.51
#Sta/Elev= 30
  4740.2  346.59  4746.8  345.76  4817.0  343.07  4885.6  342.63  4890.7  342.12
  4906.6  342.57  4918.8  342.70  4939.0  342.10  4949.2  339.81  4954.2  341.92
  4959.3  339.08  4969.4  342.42  4979.5  342.37  4989.6  338.59  4997.2  337.63
  4997.5  337.13  5001.0  337.13  5001.2  337.63  5003.8  337.63  5009.8  342.66
  5039.9  341.82  5080.1  342.62  5120.3  342.36  5130.3  342.75  5150.4  342.17
  5160.5  342.39  5170.5  343.49  5217.5  343.27  5331.2  344.95  5398.0  346.64
#Mann=5,-1,0
  4740.2    0.05       0  4906.6    0.12       0  4997.2    0.07       0
  5001.2    0.12       0  5217.5    0.05       0
Bank Sta=4997.2,5001.2
Exp/Cntr=0.3,0.1

Type RM Length L Ch R = 1,4287,291,291,291
BEGIN DESCRIPTION:
Prairie Creek Trib E4286.8
END DESCRIPTION:
XS GIS Cut Line= 3
      2702150.89      6814641.29      2701942.95      6814863.48
      2701839.17      6815367.29
#Sta/Elev= 30
  4699.5  348.53  4766.6  344.80  4827.5  342.80  4893.6  341.97  4907.8  341.36
  4915.1  340.18  4929.3  340.68  4936.1  339.20  4943.5  341.61  4950.3  337.83
  4957.6  341.80  4964.5  340.05  4971.8  341.94  5003.8  341.88  5009.9  338.58
  5013.0  335.35  5013.3  334.85  5017.0  335.35  5021.7  339.22  5031.9  341.84
  5042.1  342.31  5065.3  341.23  5166.0  340.16  5216.3  340.67  5236.1  341.83
  5261.5  341.31  5268.8  342.03  5311.8  342.90  5338.2  342.10  5518.2  346.21
#Mann=5,-1,0
  4699.5    0.05       0  4827.5    0.12       0  5013.0    0.07       0
  5017.0    0.12       0  5268.8    0.05       0
Bank Sta=5013,5017
Exp/Cntr=0.3,0.1

Type RM Length L Ch R = 1,3996,414,414,414
BEGIN DESCRIPTION:
Prairie Creek Trib E3996.148
END DESCRIPTION:
XS GIS Cut Line= 3
      2702125.99      6814611.01      2701670.96      6814810.91
      2701757.81      6815402.67
#Sta/Elev= 30
  4503.0  348.76  4607.9  344.15  4668.4  342.40  4721.4  343.10  4754.2  341.34
  4994.5  340.11  5000.0  335.25  5002.7  340.11  5020.3  335.28  5028.4  335.09
  5028.7  334.59  5032.4  335.09  5040.5  337.92  5050.6  339.58  5060.7  338.55
  5067.5  335.87  5072.5  338.74  5101.2  340.07  5111.3  339.28  5137.3  339.68
  5142.3  340.76  5182.0  339.28  5285.2  340.02  5300.0  337.98  5303.3  337.52
  5323.5  340.53  5341.6  341.31  5346.7  340.33  5384.2  342.54  5598.1  347.27
#Mann=6,-1,0
  4503.0    0.05       0  4607.9    0.12       0  5028.4    0.07       0
  5032.4    0.12       0  5285.2    0.07       0  5300.0    0.05       0
Bank Sta=5028.4,5032.4
Exp/Cntr=0.3,0.1

Type RM Length L Ch R = 1,3582,405,405,405
BEGIN DESCRIPTION:
Prairie Creek Trib E3582.31
END DESCRIPTION:
XS GIS Cut Line= 3
      2701478.27      6814150.99      2701311.53      6814861.53
      2701232.82      6815253.77
#Sta/Elev= 30
  4270.2  361.87  4341.4  357.13  4352.4  355.61  4383.2  354.58  4444.8  348.18
  4478.9  345.78  4588.6  339.76  4626.6  339.88  4653.8  338.97  4660.5  337.15
  4681.1  336.41  4711.9  338.38  4738.6  337.54  4753.0  335.69  4804.3  336.29
  4855.7  338.50  4886.5  336.95  4955.9  338.11  4968.7  337.42  4979.0  334.08
  4987.2  334.06  4987.5  333.56  4991.2  334.06  4997.2  336.99  5023.4  337.89
  5105.5  339.58  5132.1  341.03  5156.4  343.77  5244.3  345.69  5400.1  351.80
#Mann=5,-1,0
  4270.2   0.035       0  4626.6    0.12       0  4987.2    0.07       0
  4991.2    0.12       0  5023.4    0.05       0
Bank Sta=4987.2,4991.2
Exp/Cntr=0.3,0.1

Type RM Length L Ch R = 1,3177,340,340,340
BEGIN DESCRIPTION:
Prairie Creek Trib E3177.132
END DESCRIPTION:
XS GIS Cut Line= 3
      2701388.72      6813884.84      2701115.57      6814610.00
      2700964.08      6815273.63
#Sta/Elev= 30
  4225.1  356.04  4242.0  356.34  4307.8  353.67  4327.3  354.89  4355.7  354.47
  4459.4  351.55  4642.1  343.32  4753.8  339.65  4814.6  338.92  4984.8  337.22
  5003.1  335.04  5009.3  331.57  5009.5  331.07  5013.3  331.57  5018.5  334.72
  5023.6  333.44  5031.8  337.25  5061.5  336.56  5072.8  332.87  5103.6  336.30
  5124.1  335.70  5157.7  336.76  5185.7  335.54  5246.9  338.06  5291.8  339.63
  5334.7  343.67  5473.9  347.30  5565.2  351.15  5595.9  351.24  5680.7  348.18
#Mann=8,-1,0
  4225.1   0.035       0  4355.7    0.05       0  4459.4   0.035       0
  4642.1    0.05       0  4814.6    0.12       0  5009.3    0.07       0
  5013.3    0.12       0  5246.9    0.05       0
Bank Sta=5009.3,5013.3
Exp/Cntr=0.3,0.1

Type RM Length L Ch R = 1,2837,397,397,397
BEGIN DESCRIPTION:
Prairie Creek Trib E2836.94
END DESCRIPTION:
XS GIS Cut Line= 3
      2700857.21      6813820.85      2700849.09      6814669.26
      2700833.94      6815177.89
#Sta/Elev= 30
  4159.9  361.11  4233.1  355.68  4260.1  352.77  4280.1  352.52  4420.1  343.27
  4510.1  340.17  4610.1  339.55  4770.1  336.84  4780.1  337.47  4800.1  336.28
  4824.0  336.73  4950.1  336.63  4990.1  335.68  5000.1  334.62  5004.6  332.25
  5004.9  331.75  5008.5  331.75  5008.8  332.25  5020.1  332.39  5030.1  335.73
  5070.1  335.08  5090.1  337.23  5120.1  337.52  5142.6  338.62  5190.2  341.16
  5200.2  342.79  5282.6  345.06  5350.2  347.96  5460.3  351.22  5517.2  351.16
#Mann=6,-1,0
  4159.9    0.16       0  4233.1    0.07       0  4824.0    0.12       0
  5004.6    0.07       0  5008.8    0.12       0  5142.6    0.05       0
Bank Sta=5004.6,5008.8
Exp/Cntr=0.3,0.1

Type RM Length L Ch R = 1,2440,206,206,206
BEGIN DESCRIPTION:
Prairie Creek Trib E2440.25
END DESCRIPTION:
XS GIS Cut Line= 3
      2700697.13      6813748.02      2700565.96      6814511.34
      2700478.36      6814976.45
#Sta/Elev= 30
  4233.3  357.66  4361.9  349.17  4388.8  348.13  4419.0  345.53  4520.4  340.48
  4611.7  338.76  4672.6  336.57  4805.3  334.73  4868.5  334.52  4936.4  333.66
  4956.7  334.27  4975.0  333.29  4987.2  334.11  5027.8  334.47  5033.8  335.17
  5036.8  329.27  5037.0  328.77  5040.7  328.77  5041.0  329.27  5048.2  329.30
  5068.5  331.07  5078.7  330.70  5086.2  333.81  5091.3  334.50  5143.8  333.93
  5160.1  335.00  5239.3  337.09  5358.7  343.52  5455.2  346.44  5481.1  346.37
#Mann=7,-1,0
  4233.3    0.16       0  4361.9    0.07       0  4388.8    0.05       0
  4868.5    0.12       0  5036.8    0.07       0  5041.0    0.12       0
  5239.3    0.05       0
Bank Sta=5036.8,5041
Exp/Cntr=0.3,0.1

Type RM Length L Ch R = 1,2234,539,539,539
BEGIN DESCRIPTION:
Prairie Creek Trib E2234.33
END DESCRIPTION:
XS GIS Cut Line= 3
      2700536.69      6813527.96      2700375.72      6814472.41
      2700318.55      6814897.81
#Sta/Elev= 30
  4053.1  366.42  4062.0  366.75  4144.5  362.37  4149.5  360.93  4177.9  359.80
  4218.5  355.34  4238.8  354.49  4248.9  352.90  4264.8  353.13  4284.5  350.63
  4360.5  345.74  4390.9  342.13  4418.7  341.42  4445.4  339.20  4505.6  336.87
  4626.0  334.09  4760.4  333.69  4776.4  334.34  4837.3  332.25  4959.0  334.30
  4989.5  333.55  5005.8  330.89  5006.1  330.39  5010.0  330.89  5019.8  333.95
  5070.3  332.21  5110.8  333.80  5140.9  335.69  5209.3  337.47  5440.4  345.63
#Mann=9,-1,0
  4053.1    0.07       0  4062.0    0.16       0  4284.5    0.07       0
  4418.7    0.05       0  4760.4    0.12       0  5005.8    0.07       0
  5010.0    0.12       0  5110.8    0.07       0  5209.3    0.05       0
Bank Sta=5005.8,5010
Exp/Cntr=0.3,0.1

Type RM Length L Ch R = 1,1695,639,639,639
BEGIN DESCRIPTION:
Prairie Creek Trib E1695.21
END DESCRIPTION:
XS GIS Cut Line= 3
      2700429.35      6813235.45      2700148.80      6814103.62
      2700200.71      6814896.55
#Sta/Elev= 30
  4103.5  361.51  4127.9  363.54  4191.9  365.12  4223.9  364.19  4265.7  360.14
  4271.4  360.02  4389.4  353.30  4454.7  348.45  4458.6  347.47  4477.2  347.67
  4485.4  345.87  4579.0  341.07  4609.2  338.92  4675.3  336.70  4760.9  333.42
  4939.0  331.51  4950.1  331.02  4958.4  326.31  4958.7  325.81  4962.7  326.31
  4976.3  329.84  4987.5  330.81  5086.8  330.90  5185.1  330.89  5263.8  330.81
  5394.1  336.31  5480.0  338.03  5564.4  338.29  5724.8  342.31  5810.5  343.09
#Mann=14,-1,0
  4103.5    0.07       0  4265.7    0.16       0  4271.4    0.07       0
  4389.4    0.16       0  4454.7    0.07       0  4579.0    0.16       0
  4609.2    0.07       0  4675.3    0.05       0  4958.4    0.07       0
  4962.7    0.05       0  4987.5    0.07       0  5086.8    0.05       0
  5185.1    0.07       0  5480.0    0.05       0
Bank Sta=4958.4,4962.7
Exp/Cntr=0.3,0.1

Type RM Length L Ch R = 1,1056,0,0,0
BEGIN DESCRIPTION:
Prairie Creek Trib E1055.963
END DESCRIPTION:
XS GIS Cut Line= 3
      2700351.02      6812885.97      2699575.97      6813910.92
      2700147.75      6814965.15
#Sta/Elev= 30
  3715.0  357.17  3765.0  357.53  3794.1  353.86  3879.4  349.41  3900.2  346.95
  3958.4  346.48  4131.2  342.71  4335.6  337.07  4349.7  335.60  4435.9  336.01
  4443.4  336.23  4449.6  338.37  4457.9  337.43  4464.2  334.11  4507.9  331.99
  4643.1  329.99  4772.1  329.71  4863.7  327.66  4949.9  328.05  4978.2  327.27
  4984.3  323.99  4984.6  323.49  4988.7  323.99  4996.9  326.30  5022.8  328.10
  5406.5  330.42  5870.4  330.60  6034.0  333.38  6165.2  338.95  6199.3  339.36
#Mann=5,-1,0
  3715.0    0.16       0  3958.4    0.07       0  4131.2    0.05       0
  4984.3    0.05       0  4988.7    0.05       0
Bank Sta=4984.3,4988.7
Exp/Cntr=0.3,0.1

Chan Stop Cuts=-1
