--- Purtis Creek.prj (project) ---

Proj Title=Purtis Creek Base Level Engineering
Current Plan=p01
Default Exp/Contr=0.3,0.1
English Units
Geom File=g01
Flow File=f01
Plan File=p01
BEGIN DESCRIPTION:
Purtis Creek
END DESCRIPTION:

--- Purtis Creek.p01 (plan) ---

Plan Title=Multiple Run
Short Identifier=Multiple
Geom File=g01
Flow File=f01
Subcritical Flow
K Sum by GR= 0
Std Step Tol= 0.01
Critical Tol= 0.01
Num of Std Step Trials= 20
Max Error Tol= 0.3
Flow Tol Ratio= 0.001
Split Flow NTrial= 30
Split Flow Tol= 0.02
Split Flow Ratio= 0.02
Log Output Level= 0
Friction Slope Method= 1
Unsteady Friction Slope Method= 2
Unsteady Bridges Friction Slope Method= 1
Parabolic Critical Depth
Global Vel Dist=  1 , 1 , 1
Global Log Level= 0
CheckData=True
Encroach Param= -1, 0, 0, 0
BEGIN DESCRIPTION:
Multiple Run
END DESCRIPTION:

--- Purtis Creek.f01 (steady flow) ---

Flow Title=Multiple
Number of Profiles=7
Profile Names=10-year,25-year,50-year,1pct_min,100-year,1pct_plu,500-year
River Rch & RM= Purtis Creek,Reach-1,41701
     541     726     876     526    1049    2094    1508
River Rch & RM= Purtis Creek,Reach-1,33117
     700     951    1159     701    1398    2790    2042
River Rch & RM= Purtis Creek,Reach-1,30004
    1016    1407    1735    1061    2117    4224    3162
River Rch & RM= Purtis Creek,Reach-1,27019
    1098    1523    1878    1148    2291    4572    3421
River Rch & RM= Purtis Creek,Reach-1,22931
    1645    2327    2910    1802    3595    7172    5505
River Rch & RM= Purtis Creek,Reach-1,21620
    1704    2415    3023    1874    3739    7461    5741
River Rch & RM= Purtis Creek,Reach-1,19896
    1922    2728    3417    2118    4227    8434    6489
River Rch & RM= Purtis Creek,Reach-1,14180
    1990    2826    3541    2196    4381    8742    6730
River Rch & RM= Purtis Creek,Reach-1,13353
    2140    3038    3807    2359    4707    9391    7219
River Rch & RM= Purtis Creek,Reach-1,9889
    2244    3186    3992    2474    4935    9847    7567
River Rch & RM= Purtis Creek,Reach-1,8352
    2287    3248    4071    2523    5034   10045    7723
River Rch & RM= Purtis Creek,Reach-1,7986
    2303    3272    4102    2542    5072   10121    7783
River Rch & RM= Purtis Creek,Reach-1,7640
    2288    3249    4070    2521    5029   10034    7706
River Rch & RM= Purtis Creek,Reach-1,6579
    2283    3239    4057    2512    5011    9999    7673
River Rch & RM= Purtis Creek,Reach-1,5962
    2266    3211    4017    2484    4956    9889    7571
River Rch & RM= Purtis Creek,Reach-1,4610
    3071    4391    5522    3424    6833   13633   10467
Boundary for River Rch & Prof#=Purtis Creek,Reach-1,1
Up Type=0
Dn Type=3
Dn Slope=0.005
Boundary for River Rch & Prof#=Purtis Creek,Reach-1,2
Up Type=0
Dn Type=3
Dn Slope=0.005
Boundary for River Rch & Prof#=Purtis Creek,Reach-1,3
Up Type=0
Dn Type=3
Dn Slope=0.005
Boundary for River Rch & Prof#=Purtis Creek,Reach-1,4
Up Type=0
Dn Type=3
Dn Slope=0.005
Boundary for River Rch & Prof#=Purtis Creek,Reach-1,5
Up Type=0
Dn Type=3
Dn Slope=0.005
Boundary for River Rch & Prof#=Purtis Creek,Reach-1,6
Up Type=0
Dn Type=3
Dn Slope=0.005
Boundary for River Rch & Prof#=Purtis Creek,Reach-1,7
Up Type=0
Dn Type=3
Dn Slope=0.005

--- Purtis Creek.g01 (geometry) ---

Geom Title=Existing Conditions

River Reach=Purtis Creek,Reach-1
Reach XY= 30
      2761826.00      6840161.00      2760877.58      6840157.17
      2760035.82      6839021.46      2759195.41      6838882.03
      2759473.26      6838519.24      2758283.69      6837767.47
      2758022.56      6836212.19      2757185.80      6835171.48
      2755872.99      6834855.54      2755665.54      6834261.81
      2754834.46      6834708.37      2753432.08      6833369.13
      2750862.35      6831847.81      2750276.36      6831245.84
      2750772.60      6830759.71      2750662.46      6830347.57
      2750180.89      6830255.88      2749960.84      6829761.38
      2749212.61      6830147.59      2748933.07      6829811.01
      2749118.20      6829454.79      2747836.17      6828021.32
      2746319.92      6827452.87      2745724.42      6826664.83
      2742512.79      6825647.38      2741129.29      6823709.64
      2741123.76      6822716.93      2739970.55      6820216.19
      2738870.14      6819663.07      2737476.00      6819661.00

Type RM Length L Ch R = 1,41701,100,100,100
BEGIN DESCRIPTION:
Purtis Creek41701.428
END DESCRIPTION:
XS GIS Cut Line= 3
      2761731.24      6839996.10      2761789.90      6840197.12
      2761867.33      6840427.45
#Sta/Elev= 30
  4790.6  526.22  4819.9  525.85  4837.4  525.75  4862.3  524.77  4895.7  522.85
  4901.0  522.12  4910.3  521.71  4920.7  521.95  4941.5  520.89  4962.4  521.72
  4967.9  522.51  4973.1  525.14  4983.2  524.85  4993.6  523.27  5006.4  518.01
  5012.6  517.95  5012.9  517.45  5016.4  517.45  5016.6  517.95  5032.7  521.27
  5046.3  522.08  5069.4  521.36  5127.2  521.40  5132.5  521.89  5141.2  520.06
  5158.7  522.37  5164.0  522.00  5190.2  522.84  5233.9  525.15  5243.0  525.32
#Mann=5,-1,0
  4790.6    0.16       0  4819.9    0.12       0  5012.6    0.07       0
  5016.6    0.12       0  5233.9   0.063       0
Bank Sta=5012.6,5016.6
Exp/Cntr=0.3,0.1

Type RM Length L Ch R = 1,41601,82,82,82
BEGIN DESCRIPTION:
Purtis Creek41600.76
END DESCRIPTION:
XS GIS Cut Line= 3
      2761646.26      6840072.50      2761718.62      6840268.06
      2761809.34      6840464.07
#Sta/Elev= 30
  4791.2  524.54  4810.6  524.49  4835.6  524.53  4891.1  522.25  4896.4  522.90
  4921.5  521.47  4960.2  520.73  4970.9  521.32  4992.2  521.44  5006.9  520.45
  5014.0  519.15  5022.3  518.48  5022.6  517.98  5026.1  517.98  5026.3  518.48
  5029.8  519.47  5036.0  520.39  5047.0  520.86  5052.8  521.71  5058.3  521.81
  5069.1  520.79  5081.2  520.58  5113.1  521.42  5121.5  521.25  5135.2  521.92
  5144.5  521.73  5163.9  522.62  5172.9  522.88  5195.8  526.84  5215.7  527.31
#Mann=5,-1,0
  4791.2    0.16       0  4810.6    0.12       0  5022.3    0.07       0
  5026.3    0.12       0  5163.9   0.063       0
Bank Sta=5022.3,5026.3
Exp/Cntr=0.3,0.1

Type RM Length L Ch R = 1,41519,109,109,109
BEGIN DESCRIPTION:
Purtis Creek41518.59
END DESCRIPTION:
XS GIS Cut Line= 3
      2761554.49      6840071.40      2761661.16      6840327.27
      2761748.36      6840515.54
#Sta/Elev= 30
  4723.4  524.35  4739.8  523.00  4760.3  523.09  4763.6  523.00  4769.0  524.53
  4777.1  524.62  4787.4  522.00  4792.9  522.94  4798.8  520.74  4816.7  519.57
  4822.1  520.59  4840.5  519.26  4853.0  520.23  4875.8  520.03  4917.4  520.09
  4922.8  521.27  4939.7  520.86  4946.7  519.43  4975.9  521.01  4983.0  519.84
  4991.8  517.09  4992.1  516.59  4995.8  517.09  4999.7  519.64  5022.6  520.58
  5074.5  520.62  5097.3  520.55  5159.0  522.71  5206.4  527.46  5208.1  527.46
#Mann=8,-1,0
  4723.4    0.16       0  4760.3    0.12       0  4875.8    0.16       0
  4991.8    0.07       0  4995.8    0.16       0  5074.5    0.12       0
  5097.3   0.063       0  5206.4    0.05       0
Bank Sta=4991.8,4995.8
Exp/Cntr=0.3,0.1

Type RM Length L Ch R = 1,41410,124,124,124
BEGIN DESCRIPTION:
Purtis Creek41409.57
END DESCRIPTION:
XS GIS Cut Line= 3
      2761520.92      6840061.18      2761563.90      6840361.69
      2761578.44      6840516.44
#Sta/Elev= 30
  4696.8  525.27  4716.8  524.18  4737.0  524.07  4748.6  522.98  4765.1  520.47
  4770.2  520.63  4777.4  519.72  4787.5  519.24  4807.7  518.98  4858.2  519.94
  4880.1  519.14  4911.5  519.90  4959.3  519.15  4977.1  520.30  4989.6  520.35
  5002.5  519.90  5009.7  519.07  5017.8  517.24  5018.0  516.74  5021.5  516.74
  5021.8  517.24  5029.8  519.45  5049.9  519.83  5075.6  523.42  5080.7  522.26
  5090.1  523.45  5120.2  524.75  5140.3  524.96  5149.3  525.98  5155.8  527.25
#Mann=6,-1,0
  4696.8    0.16       0  4748.6    0.12       0  4880.1    0.16       0
  5017.8    0.07       0  5021.8    0.16       0  5149.3   0.063       0
Bank Sta=5017.8,5021.8
Exp/Cntr=0.3,0.1

Type RM Length L Ch R = 1,41286,135,135,135
BEGIN DESCRIPTION:
Purtis Creek41285.83
END DESCRIPTION:
XS GIS Cut Line= 3
      2761456.17      6840111.22      2761439.86      6840365.15
      2761439.15      6840506.49
#Sta/Elev= 30
  4749.4  524.89  4759.2  524.76  4763.5  523.53  4789.3  517.07  4799.3  516.24
  4809.3  518.34  4827.2  518.57  4859.4  517.75  4869.4  518.84  4909.5  518.27
  4919.5  518.86  4928.5  518.84  4939.6  518.81  4959.6  519.56  4969.6  518.11
  4977.7  515.95  4977.9  515.45  4981.4  515.45  4981.7  515.95  4985.4  517.95
  4990.4  517.14  4999.3  519.27  5019.7  519.50  5029.7  520.60  5039.7  520.77
  5049.7  521.69  5059.7  523.44  5069.7  523.56  5119.7  525.63  5145.2  527.23
#Mann=5,-1,0
  4749.4    0.16       0  4763.5    0.12       0  4928.5    0.16       0
  4977.7    0.07       0  4981.7    0.16       0
Bank Sta=4977.7,4981.7
Exp/Cntr=0.3,0.1

Type RM Length L Ch R = 1,41151,80,80,80
BEGIN DESCRIPTION:
Purtis Creek41150.64
END DESCRIPTION:
XS GIS Cut Line= 6
      2761396.36      6840116.23      2761363.59      6840255.05
      2761318.00      6840316.71      2761292.06      6840363.70
      2761280.49      6840424.03      2761294.75      6840554.30
#Sta/Elev= 30
  4784.7  523.32  4799.9  523.41  4805.4  522.79  4811.7  522.34  4820.4  517.66
  4830.7  516.68  4854.0  517.02  4871.8  518.64  4882.1  519.05  4910.1  518.29
  4936.3  517.92  4981.4  518.43  5001.4  517.72  5009.5  517.96  5020.4  516.45
  5020.7  515.95  5024.2  515.95  5024.4  516.45  5031.9  517.57  5038.5  517.83
  5066.9  517.08  5106.0  517.56  5113.8  518.41  5136.3  519.09  5198.8  524.70
  5206.7  525.21  5218.8  524.59  5226.9  525.10  5236.9  527.76  5250.3  528.33
#Mann=6,-1,0
  4784.7    0.16       0  4805.4    0.12       0  4910.1    0.16       0
  5020.4    0.07       0  5024.4    0.16       0  5198.8   0.063       0
Bank Sta=5020.4,5024.4
Exp/Cntr=0.3,0.1

Type RM Length L Ch R = 1,41071,126,126,126
BEGIN DESCRIPTION:
Purtis Creek41070.94
END DESCRIPTION:
XS GIS Cut Line= 6
      2761293.49      6840080.19      2761296.32      6840189.54
      2761268.85      6840261.39      2761219.57      6840361.93
      2761215.20      6840427.85      2761223.78      6840526.28
#Sta/Elev= 30
  4756.9  524.94  4777.7  524.99  4817.7  523.75  4847.7  522.01  4857.7  521.12
  4864.5  519.98  4869.7  519.98  4889.3  518.06  4907.3  516.99  4932.0  517.18
  4937.3  516.74  4959.1  516.56  4974.2  517.15  4983.6  511.59  4983.9  511.09
  4987.4  511.09  4987.6  511.59  4998.2  512.47  5001.1  516.18  5011.3  517.01
  5044.0  516.82  5050.8  517.19  5057.9  516.81  5064.9  518.60  5074.9  519.98
  5135.1  521.33  5195.8  525.10  5205.4  526.35  5215.4  526.69  5220.7  526.02
#Mann=4,-1,0
  4756.9    0.16       0  4983.6    0.07       0  4987.6    0.16       0
  5195.8   0.063       0
Bank Sta=4983.6,4987.6
Exp/Cntr=0.3,0.1

Type RM Length L Ch R = 1,40945,92,92,92
BEGIN DESCRIPTION:
Purtis Creek40945.14
END DESCRIPTION:
XS GIS Cut Line= 3
      2761214.69      6840090.67      2761171.17      6840218.41
      2761105.42      6840447.72
#Sta/Elev= 30
  4866.0  524.24  4879.8  524.20  4887.5  523.55  4898.0  521.34  4905.9  520.05
  4919.2  518.63  4950.9  516.31  4961.4  516.30  4973.9  515.45  5005.2  516.64
  5014.0  516.05  5022.4  511.00  5022.7  510.50  5026.2  510.50  5026.4  511.00
  5033.7  514.55  5038.9  516.14  5045.3  516.43  5077.9  515.93  5097.3  516.49
  5111.6  516.45  5138.9  517.45  5145.4  518.01  5179.1  518.96  5184.3  518.86
  5201.3  519.80  5218.1  521.26  5223.3  520.84  5232.5  520.74  5239.5  521.25
#Mann=3,-1,0
  4866.0    0.16       0  5022.4    0.07       0  5026.4    0.16       0
Bank Sta=5022.4,5026.4
Exp/Cntr=0.3,0.1

Type RM Length L Ch R = 1,40853,94,94,94
BEGIN DESCRIPTION:
Purtis Creek40853.28
END DESCRIPTION:
XS GIS Cut Line= 3
      2761089.54      6840101.73      2761081.31      6840212.97
      2761050.30      6840437.79
#Sta/Elev= 30
  4890.2  523.30  4899.5  523.20  4919.6  522.17  4929.6  521.89  4939.6  521.33
  4959.7  519.73  4969.7  518.00  4989.7  515.74  4998.3  511.13  5001.7  511.13
  5002.4  510.54  5002.7  510.04  5006.2  510.04  5006.4  510.54  5009.9  516.01
  5019.9  515.80  5030.0  515.18  5040.1  515.33  5050.2  515.83  5060.3  515.08
  5070.4  515.62  5081.4  515.53  5090.6  515.91  5110.8  516.25  5171.4  518.05
  5181.5  518.47  5191.6  519.65  5211.7  519.94  5225.2  520.49  5228.7  521.22
#Mann=3,-1,0
  4890.2    0.16       0  5002.4    0.07       0  5006.4    0.16       0
Bank Sta=5002.4,5006.4
Exp/Cntr=0.3,0.1

Type RM Length L Ch R = 1,40759,77,77,77
BEGIN DESCRIPTION:
Purtis Creek40759.02
END DESCRIPTION:
XS GIS Cut Line= 3
      2761005.52      6840083.38      2760996.60      6840184.92
      2760986.78      6840437.50
#Sta/Elev= 30
  4901.0  522.39  4908.7  521.93  4922.4  521.65  4928.7  521.38  4938.8  520.60
  4953.2  520.25  4958.8  519.44  4968.9  515.89  4976.9  509.78  4977.2  509.28
  4980.7  509.28  4980.9  509.78  4998.5  510.02  5009.0  509.89  5029.0  510.68
  5039.0  510.10  5049.0  512.28  5059.1  515.72  5079.1  515.49  5089.1  515.06
  5119.1  515.37  5129.1  515.91  5145.6  516.47  5150.6  516.34  5159.1  516.87
  5169.1  517.00  5199.2  518.01  5219.2  519.22  5249.2  520.40  5255.7  520.84
#Mann=4,-1,0
  4901.0    0.12       0  4922.4    0.16       0  4976.9    0.07       0
  4980.9    0.16       0
Bank Sta=4976.9,4980.9
Exp/Cntr=0.3,0.1

Type RM Length L Ch R = 1,40682,92,92,92
BEGIN DESCRIPTION:
Purtis Creek40681.59
END DESCRIPTION:
XS GIS Cut Line= 3
      2760935.02      6840037.27      2760925.45      6840165.86
      2760897.97      6840426.06
#Sta/Elev= 30
  4875.9  521.16  4889.7  521.15  4919.8  519.76  4927.4  519.63  4939.8  518.87
  4941.7  518.95  4949.8  519.31  4959.9  518.76  4969.9  517.92  4979.9  517.73
  4989.9  516.69  4999.9  511.18  5004.8  511.18  5008.0  509.49  5008.3  508.99
  5011.8  508.99  5012.0  509.49  5020.1  514.37  5040.2  514.61  5046.2  514.93
  5060.3  514.69  5100.5  515.44  5110.6  514.91  5139.1  515.21  5144.1  515.04
  5211.1  516.59  5237.1  517.66  5242.0  517.48  5251.4  517.73  5266.5  518.61
#Mann=5,-1,0
  4875.9    0.12       0  4941.7    0.16       0  5008.0    0.07       0
  5012.0    0.16       0  5237.1   0.035       0
Bank Sta=5008,5012
Exp/Cntr=0.3,0.1

Type RM Length L Ch R = 1,40590,147,147,147
BEGIN DESCRIPTION:
Purtis Creek40590.35
END DESCRIPTION:
XS GIS Cut Line= 3
      2760898.41      6839859.94      2760844.35      6840132.70
      2760797.57      6840423.80
#Sta/Elev= 30
  4724.4  520.96  4756.1  519.42  4766.9  518.32  4786.6  517.65  4796.8  516.26
  4807.0  516.28  4813.0  515.17  4818.1  515.19  4827.4  513.40  4837.6  515.44
  4864.2  517.49  4880.0  514.16  4888.6  512.98  4909.0  512.66  4920.6  512.79
  4939.6  514.17  4949.8  513.52  4980.3  514.04  4990.5  510.73  4997.1  509.90
  4997.3  509.40  5000.8  509.40  5001.1  509.90  5019.8  514.17  5061.5  513.56
  5142.5  515.03  5162.8  514.81  5233.7  516.05  5292.6  518.20  5297.3  518.24
#Mann=5,-1,0
  4724.4    0.12       0  4880.0    0.16       0  4997.1    0.07       0
  5001.1    0.16       0  5292.6   0.035       0
Bank Sta=4997.1,5001.1
Exp/Cntr=0.3,0.1

Type RM Length L Ch R = 1,40443,156,156,156
BEGIN DESCRIPTION:
Purtis Creek40442.63
END DESCRIPTION:
XS GIS Cut Line= 3
      2760825.17      6839745.21      2760717.07      6840065.95
      2760632.16      6840317.86
#Sta/Elev= 30
  4664.1  527.85  4676.3  526.40  4701.9  524.67  4723.0  517.58  4744.6  512.94
  4765.2  513.33  4776.0  512.43  4807.5  511.85  4817.9  512.32  4833.7  511.49
  4862.6  512.37  4870.7  511.57  4881.3  511.36  4902.4  512.45  4912.9  511.91
  4922.9  512.34  4944.6  512.08  4959.7  513.03  4976.2  512.37  4991.2  512.59
  4995.3  509.03  4995.6  508.53  4999.1  508.53  4999.3  509.03  5002.6  509.03
  5007.9  511.61  5017.4  512.72  5036.0  513.38  5166.2  514.88  5268.4  518.57
#Mann=5,-1,0
  4664.1    0.12       0  4862.6    0.16       0  4995.3    0.07       0
  4999.3    0.16       0  5036.0    0.07       0
Bank Sta=4995.3,4999.3
Exp/Cntr=0.3,0.1

Type RM Length L Ch R = 1,40287,284,284,284
BEGIN DESCRIPTION:
Purtis Creek40287.12
END DESCRIPTION:
XS GIS Cut Line= 3
      2760785.00      6839629.93      2760626.03      6839958.51
      2760522.65      6840220.97
#Sta/Elev= 30
  4639.8  526.21  4647.8  525.46  4653.3  523.27  4670.4  523.04  4675.9  520.31
  4692.9  520.03  4698.5  517.50  4715.5  516.42  4721.1  515.09  4738.1  514.67
  4743.7  513.32  4760.7  512.67  4766.3  511.59  4811.4  510.25  4918.7  511.50
  4924.4  510.44  4930.0  511.37  4940.9  510.91  4952.5  511.60  4957.7  510.88
  4967.6  509.19  4967.8  508.69  4971.3  508.69  4971.6  509.19  4985.4  511.05
  5003.4  511.91  5021.1  511.51  5099.6  512.91  5150.9  513.09  5286.9  516.86
#Mann=5,-1,0
  4639.8    0.12       0  4957.7    0.16       0  4967.6    0.07       0
  4971.6    0.16       0  5150.9    0.07       0
Bank Sta=4967.6,4971.6
Exp/Cntr=0.3,0.1

Type RM Length L Ch R = 1,40003,259,259,259
BEGIN DESCRIPTION:
Purtis Creek40003.32
END DESCRIPTION:
XS GIS Cut Line= 3
      2760606.21      6839401.87      2760556.86      6839692.87
      2760455.91      6840167.29
#Sta/Elev= 30
  4705.6  520.44  4733.4  519.40  4755.4  516.41  4765.6  514.12  4775.7  512.58
  4806.1  510.73  4867.0  509.39  4927.9  509.37  4968.4  510.06  4974.8  509.95
  4986.7  508.75  4987.0  508.25  4990.5  508.25  4990.7  508.75  5026.7  509.58
  5039.7  509.09  5070.4  510.33  5081.4  511.43  5101.1  511.97  5111.3  511.55
  5125.8  512.05  5171.7  511.92  5175.4  512.40  5203.3  512.31  5225.0  513.32
  5274.9  514.27  5309.3  514.46  5363.5  514.26  5457.6  515.76  5485.8  516.73
#Mann=5,-1,0
  4705.6    0.12       0  4986.7    0.07       0  4990.7    0.12       0
  5171.7   0.063       0  5309.3   0.035       0
Bank Sta=4986.7,4990.7
Exp/Cntr=0.3,0.1

Type RM Length L Ch R = 1,39744,62,62,62
BEGIN DESCRIPTION:
Purtis Creek39744.02
END DESCRIPTION:
XS GIS Cut Line= 3
      2760473.76      6839200.59      2760465.48      6839464.49
      2760467.99      6839736.64
#Sta/Elev= 30
  4737.4  519.69  4777.8  518.75  4797.8  517.45  4817.9  516.60  4837.9  514.86
  4847.9  513.38  4857.9  512.65  4897.9  510.23  4917.9  509.53  4937.9  508.36
  4977.9  507.91  5007.9  508.31  5015.9  507.70  5016.2  507.20  5019.7  507.20
  5019.9  507.70  5027.9  508.25  5041.4  508.55  5047.9  508.83  5067.9  508.75
  5077.9  509.13  5097.9  508.11  5117.9  508.94  5137.9  508.99  5158.0  509.63
  5178.0  510.76  5198.0  512.40  5228.0  513.59  5268.0  514.18  5273.6  513.95
#Mann=4,-1,0
  4737.4   0.035       0  5015.9   0.035       0  5019.9   0.035       0
  5041.4   0.063       0
Bank Sta=5015.9,5019.9
Exp/Cntr=0.3,0.1

Type RM Length L Ch R = 1,39682,128,128,128
BEGIN DESCRIPTION:
Purtis Creek39682.24
END DESCRIPTION:
XS GIS Cut Line= 3
      2760403.77      6839133.91      2760403.99      6839462.98
      2760396.48      6839695.49
#Sta/Elev= 30
  4672.9  516.25  4690.0  516.15  4720.0  515.11  4740.0  513.39  4760.0  512.13
  4800.0  511.74  4830.0  510.68  4860.0  509.04  4870.0  508.76  4940.0  507.30
  4960.0  507.57  4990.0  507.63  4998.5  506.91  5008.0  506.88  5008.2  506.38
  5011.7  506.38  5012.0  506.88  5020.0  507.49  5030.0  507.61  5040.0  508.14
  5050.0  507.98  5060.0  508.08  5080.0  509.14  5089.8  509.43  5100.0  510.12
  5130.1  511.41  5150.1  512.05  5190.1  512.67  5210.1  513.57  5234.6  513.57
#Mann=3,-1,0
  4672.9    0.16       0  5008.0    0.07       0  5012.0    0.16       0
Bank Sta=5008,5012
Exp/Cntr=0.3,0.1

Type RM Length L Ch R = 1,39554,120,120,120
BEGIN DESCRIPTION:
Purtis Creek39553.58
END DESCRIPTION:
XS GIS Cut Line= 3
      2760358.95      6839067.51      2760303.36      6839388.68
      2760241.73      6839731.34
#Sta/Elev= 30
  4674.7  512.92  4717.5  512.88  4722.6  512.02  4739.1  512.37  4759.4  512.08
  4803.7  507.86  4837.1  506.72  4842.1  506.15  4881.2  506.01  4894.8  505.63
  4895.1  505.13  4898.6  505.13  4898.8  505.63  4911.7  506.06  4999.3  506.94
  5033.5  506.16  5053.8  507.81  5064.0  508.15  5069.8  508.91  5094.4  510.35
  5104.6  512.02  5114.8  513.17  5127.1  513.43  5145.2  513.38  5187.2  512.11
  5226.5  511.77  5318.0  513.37  5328.1  514.08  5338.3  513.68  5348.8  513.73
#Mann=5,-1,0
  4674.7    0.05       0  4803.7    0.16       0  4894.8    0.07       0
  4898.8    0.16       0  5127.1    0.05       0
Bank Sta=4894.8,4898.8
Exp/Cntr=0.3,0.1

Type RM Length L Ch R = 1,39434,310,310,310
BEGIN DESCRIPTION:
Purtis Creek39433.6
END DESCRIPTION:
XS GIS Cut Line= 3
      2760313.16      6838966.60      2760199.40      6839337.91
      2760134.71      6839556.59
#Sta/Elev= 30
  4614.0  511.72  4617.7  511.72  4622.6  510.84  4655.4  510.82  4660.6  510.16
  4688.1  510.05  4693.3  509.54  4712.7  509.17  4726.1  507.88  4744.1  507.77
  4775.5  506.83  4791.6  506.09  4796.8  505.34  4806.9  505.15  4838.2  505.15
  4857.1  505.85  4993.4  506.13  5006.6  506.10  5014.0  504.80  5014.2  504.30
  5017.7  504.30  5018.0  504.80  5031.8  506.97  5057.7  507.35  5098.3  508.94
  5103.6  508.57  5130.7  510.06  5142.0  509.68  5170.1  511.16  5230.4  511.74
#Mann=3,-1,0
  4614.0    0.05       0  5014.0    0.05       0  5018.0    0.05       0
Bank Sta=5014,5018
Exp/Cntr=0.3,0.1

Type RM Length L Ch R = 1,39124,175,175,175
BEGIN DESCRIPTION:
Purtis Creek39123.59
END DESCRIPTION:
XS GIS Cut Line= 3
      2760083.06      6838912.94      2760084.70      6839071.44
      2760075.53      6839357.09
#Sta/Elev= 30
  4844.0  507.29  4862.1  504.56  4872.1  504.21  4882.1  504.09  4892.1  503.76
  4902.1  503.61  4922.1  503.73  4932.1  503.19  4940.1  502.45  4940.3  501.95
  4943.8  501.95  4944.1  502.45  4952.1  502.63  4962.1  503.18  4972.1  503.25
  4982.1  502.52  4992.1  502.71  5004.8  502.66  5032.1  504.21  5042.1  504.41
  5062.1  505.25  5072.1  505.53  5117.5  506.36  5122.5  506.81  5142.1  507.50
  5172.2  508.01  5182.2  508.31  5192.2  508.38  5252.2  509.54  5288.3  509.85
#Mann=3,-1,0
  4844.0    0.05       0  4940.1    0.05       0  4944.1    0.05       0
Bank Sta=4940.1,4944.1
Exp/Cntr=0.3,0.1

Type RM Length L Ch R = 1,38949,151,151,151
BEGIN DESCRIPTION:
Purtis Creek38949.06
END DESCRIPTION:
XS GIS Cut Line= 3
      2759932.22      6838907.95      2759931.86      6839013.16
      2759929.67      6839283.24
#Sta/Elev= 30
  4897.4  508.27  4901.4  508.27  4910.4  505.95  4930.4  504.80  4940.4  504.41
  4970.4  503.64  4990.4  502.68  4997.0  501.33  4997.3  500.83  5000.8  500.83
  5001.0  501.33  5002.6  501.33  5010.4  502.53  5020.4  502.54  5030.4  502.76
  5040.4  503.32  5050.4  503.43  5070.4  503.12  5080.5  503.23  5107.0  504.00
  5112.0  503.90  5120.5  504.16  5130.5  504.21  5160.5  505.26  5170.5  505.84
  5180.5  506.78  5210.5  508.76  5220.5  509.16  5240.5  509.36  5272.7  508.93
#Mann=3,-1,0
  4897.4    0.05       0  4997.0    0.05       0  5001.0    0.05       0
Bank Sta=4997,5001
Exp/Cntr=0.3,0.1

Type RM Length L Ch R = 1,38798,136,136,136
BEGIN DESCRIPTION:
Purtis Creek38798.35
END DESCRIPTION:
XS GIS Cut Line= 3
      2759795.90      6838850.10      2759797.31      6839063.13
      2759794.13      6839327.67
#Sta/Elev= 30
  4788.8  512.74  4799.7  512.88  4809.7  512.65  4819.7  511.86  4849.7  511.68
  4899.7  508.47  4909.7  507.69  4919.7  506.63  4939.7  505.15  4949.7  504.19
  4969.7  503.02  4979.7  502.83  4989.7  501.85  4998.3  502.41  5001.8  502.41
  5009.7  501.15  5017.7  501.07  5018.0  500.57  5021.5  500.57  5021.7  501.07
  5029.7  501.85  5059.7  502.75  5069.7  503.26  5089.7  503.84  5129.7  505.37
  5139.7  505.49  5179.7  506.59  5209.7  508.12  5219.7  508.84  5266.4  511.00
#Mann=3,-1,0
  4788.8    0.05       0  5017.7    0.05       0  5021.7    0.05       0
Bank Sta=5017.7,5021.7
Exp/Cntr=0.3,0.1

Type RM Length L Ch R = 1,38662,143,143,143
BEGIN DESCRIPTION:
Purtis Creek38662.49
END DESCRIPTION:
XS GIS Cut Line= 3
      2759668.03      6838791.42      2759661.37      6839064.03
      2759660.52      6839277.84
#Sta/Elev= 30
  4730.3  509.02  4749.9  507.76  4759.9  507.69  4769.9  508.15  4779.9  507.85
  4799.9  507.87  4849.9  505.63  4889.9  502.82  4919.9  501.71  4939.9  501.40
  4959.9  501.60  4970.0  501.47  4980.0  500.32  4990.0  497.75  4997.0  496.88
  4997.2  496.38  5000.7  496.38  5001.0  496.88  5003.0  496.88  5010.0  498.51
  5020.0  498.67  5030.0  499.85  5040.0  501.74  5070.0  501.41  5110.0  502.03
  5150.0  504.24  5180.0  506.63  5200.0  509.29  5210.0  510.27  5216.8  511.55
#Mann=3,-1,0
  4730.3    0.05       0  4997.0    0.05       0  5001.0    0.05       0
Bank Sta=4997,5001
Exp/Cntr=0.3,0.1

Type RM Length L Ch R = 1,38519,219,219,219
BEGIN DESCRIPTION:
Purtis Creek38519.43
END DESCRIPTION:
XS GIS Cut Line= 3
      2759597.22      6838743.40      2759517.79      6839063.56
      2759539.91      6839326.87
#Sta/Elev= 30
  4672.6  506.83  4690.7  506.16  4702.3  505.09  4721.6  504.58  4743.7  503.16
  4835.0  502.54  4845.3  502.11  4855.6  501.25  4896.8  500.30  4945.4  501.28
  4968.9  501.11  4979.2  497.94  4984.7  495.73  4985.0  495.23  4988.5  495.23
  4988.7  495.73  4991.9  496.21  5002.5  496.19  5009.9  499.18  5037.9  500.63
  5090.2  501.58  5110.3  502.32  5150.4  504.41  5190.6  507.60  5210.6  508.08
  5220.7  508.02  5240.7  508.94  5250.8  513.76  5260.8  514.69  5266.7  512.77
#Mann=3,-1,0
  4672.6    0.05       0  4984.7    0.05       0  4988.7    0.05       0
Bank Sta=4984.7,4988.7
Exp/Cntr=0.3,0.1

Type RM Length L Ch R = 1,38300,101,101,101
BEGIN DESCRIPTION:
Purtis Creek38299.97
END DESCRIPTION:
XS GIS Cut Line= 3
      2759576.96      6838671.42      2759426.37      6838926.24
      2759333.76      6839109.69
#Sta/Elev= 30
  4704.1  506.96  4749.7  504.09  4777.0  500.60  4792.6  501.72  4878.4  499.84
  4946.7  500.97  4957.2  493.09  4957.4  492.59  4961.2  493.09  4968.2  494.86
  4974.0  499.60  4984.4  496.74  4989.6  494.27  4995.4  498.30  5000.0  494.74
  5005.6  494.74  5017.1  498.84  5039.4  500.84  5050.2  500.77  5056.1  498.08
  5072.6  496.47  5078.4  499.26  5084.0  496.65  5095.0  497.00  5100.7  497.85
  5106.3  504.26  5113.4  505.14  5128.6  508.86  5139.7  509.34  5205.6  509.12
#Mann=5,-1,0
  4704.1    0.05       0  4957.2    0.07       0  4961.2    0.05       0
  4984.4    0.16       0  5113.4    0.05       0
Bank Sta=4957.2,4961.2
Exp/Cntr=0.3,0.1

Type RM Length L Ch R = 1,38199,243,243,243
BEGIN DESCRIPTION:
Purtis Creek38199.18
END DESCRIPTION:
XS GIS Cut Line= 3
      2759531.69      6838702.89      2759378.98      6838864.15
      2759250.67      6839033.30
#Sta/Elev= 30
  4783.2  500.91  4785.8  499.40  4793.1  499.55  4828.3  498.42  4870.8  499.22
  4877.7  498.87  4962.6  499.24  4963.3  498.63  4969.9  492.84  4976.8  493.57
  4984.1  492.82  4990.9  499.89  4998.2  499.46  5003.8  496.68  5013.1  494.50
  5017.3  492.73  5017.6  492.23  5021.1  492.23  5021.3  492.73  5026.4  493.28
  5033.9  500.02  5069.3  500.68  5076.7  499.01  5119.2  500.55  5140.0  503.35
  5150.3  505.70  5162.8  508.33  5169.1  508.56  5183.7  508.93  5217.6  507.81
#Mann=5,-1,0
  4783.2    0.05       0  4963.3    0.16       0  5017.3    0.07       0
  5021.3    0.16       0  5150.3    0.05       0
Bank Sta=5017.3,5021.3
Exp/Cntr=0.3,0.1

Type RM Length L Ch R = 1,37956,190,190,190
BEGIN DESCRIPTION:
Purtis Creek37955.87
END DESCRIPTION:
XS GIS Cut Line= 3
      2759542.73      6838673.43      2759176.54      6838853.91
      2759010.92      6838911.51
#Sta/Elev= 30
  4592.5  503.32  4596.4  501.84  4601.9  501.41  4611.1  499.45  4641.3  498.07
  4648.0  498.21  4663.7  497.74  4773.0  497.82  4888.3  497.92  4923.3  498.55
  4938.8  498.29  4967.9  499.12  4990.2  498.54  4998.3  497.59  5003.7  497.59
  5006.9  492.13  5010.2  491.98  5010.4  491.48  5013.9  491.48  5014.2  491.98
  5022.5  495.91  5038.0  498.19  5043.7  499.50  5069.1  500.30  5086.0  501.49
  5126.0  503.15  5157.1  506.24  5162.4  506.17  5170.7  506.90  5176.1  507.89
#Mann=5,-1,0
  4592.5    0.12       0  4648.0    0.05       0  4773.0    0.16       0
  5010.2    0.07       0  5014.2    0.16       0
Bank Sta=5010.2,5014.2
Exp/Cntr=0.3,0.1

Type RM Length L Ch R = 1,37766,412,412,412
BEGIN DESCRIPTION:
Purtis Creek37765.64
END DESCRIPTION:
XS GIS Cut Line= 3
      2759556.38      6838640.21      2759248.56      6838686.81
      2759056.04      6838711.34
#Sta/Elev= 30
  4689.5  505.65  4710.1  503.49  4726.7  499.11  4750.6  497.52  4882.0  497.05
  4892.2  495.70  4902.3  497.35  4912.4  497.87  4922.5  497.44  4928.1  495.97
  4933.1  497.93  4986.8  497.30  4996.9  497.48  4999.6  494.31  5004.6  494.31
  5011.5  490.27  5011.7  489.77  5015.2  489.77  5015.5  490.27  5023.6  496.87
  5033.7  497.89  5053.8  497.16  5063.9  497.36  5071.2  498.30  5104.2  497.81
  5124.4  498.94  5151.1  501.67  5156.1  501.39  5174.8  504.39  5194.9  506.12
#Mann=4,-1,0
  4689.5    0.12       0  4986.8    0.16       0  5011.5    0.07       0
  5015.5    0.16       0
Bank Sta=5011.5,5015.5
Exp/Cntr=0.3,0.1

Type RM Length L Ch R = 1,37354,188,188,188
BEGIN DESCRIPTION:
Purtis Creek37354.39
END DESCRIPTION:
XS GIS Cut Line= 3
      2759504.69      6838349.11      2759385.98      6838473.47
      2759151.74      6838634.02
#Sta/Elev= 30
  4829.6  507.38  4837.0  508.08  4844.3  504.86  4851.2  505.33  4858.4  501.99
  4865.3  502.33  4872.6  499.32  4879.5  499.44  4886.7  498.03  4893.6  498.36
  4900.9  497.06  4907.8  496.99  4922.0  494.02  4950.3  495.39  4992.7  494.91
  4997.9  493.72  5003.8  493.72  5011.6  487.92  5011.9  487.42  5015.6  487.92
  5021.7  493.68  5027.7  497.20  5046.2  497.38  5122.7  496.67  5147.6  498.03
  5159.1  498.67  5195.0  497.22  5251.8  498.08  5272.8  499.81  5285.5  499.92
#Mann=5,-1,0
  4829.6    0.16       0  5011.6    0.07       0  5015.6    0.16       0
  5046.2    0.12       0  5147.6    0.16       0
Bank Sta=5011.6,5015.6
Exp/Cntr=0.3,0.1

Type RM Length L Ch R = 1,37166,165,165,165
BEGIN DESCRIPTION:
Purtis Creek37166.02
END DESCRIPTION:
XS GIS Cut Line= 3
      2759359.31      6838211.75      2759241.04      6838362.13
      2759090.51      6838543.62
#Sta/Elev= 30
  4811.1  502.11  4820.5  502.11  4826.9  501.17  4835.0  501.31  4841.3  500.74
  4855.8  500.49  4876.6  498.39  4926.3  496.11  4948.8  495.75  4954.0  494.95
  4962.8  493.58  4969.6  488.11  4974.0  485.67  4974.3  485.17  4977.8  485.17
  4978.0  485.67  4984.1  489.44  4990.5  490.81  4998.5  493.45  5002.4  493.45
  5012.8  494.89  5047.9  494.61  5076.6  493.78  5097.4  495.71  5118.2  496.65
  5146.9  495.61  5154.7  495.82  5227.1  500.37  5232.9  500.54  5238.2  501.37
#Mann=5,-1,0
  4811.1    0.16       0  4954.0    0.12       0  4974.0    0.07       0
  4978.0    0.12       0  5227.1    0.16       0
Bank Sta=4974,4978
Exp/Cntr=0.3,0.1

Type RM Length L Ch R = 1,37001,273,273,273
BEGIN DESCRIPTION:
Purtis Creek37000.62
END DESCRIPTION:
XS GIS Cut Line= 3
      2759289.39      6838051.57      2759116.89      6838256.49
      2758994.15      6838410.63
#Sta/Elev= 30
  4735.1  500.58  4758.8  499.76  4800.5  496.94  4900.6  495.24  4907.1  494.35
  4921.4  493.93  4947.3  494.07  4956.6  494.48  4964.3  491.98  4976.6  484.87
  4976.9  484.37  4980.4  484.37  4980.6  484.87  4985.1  487.44  4992.9  493.21
  5007.7  493.39  5013.8  492.48  5028.2  493.71  5049.0  493.39  5057.0  492.64
  5077.8  492.67  5092.2  497.23  5106.7  500.43  5113.1  501.29  5121.1  503.64
  5127.5  504.44  5135.5  505.28  5156.3  505.87  5181.7  505.13  5200.0  504.52
#Mann=5,-1,0
  4735.1    0.16       0  4947.3    0.12       0  4976.6    0.07       0
  4980.6    0.12       0  5181.7    0.16       0
Bank Sta=4976.6,4980.6
Exp/Cntr=0.3,0.1

Type RM Length L Ch R = 1,36728,189,189,189
BEGIN DESCRIPTION:
Purtis Creek36727.6
END DESCRIPTION:
XS GIS Cut Line= 3
      2758999.43      6837868.61      2758968.27      6838061.81
      2758943.99      6838274.23
#Sta/Elev= 30
  4805.5  497.63  4818.0  497.42  4828.2  496.72  4856.0  496.10  4861.0  495.00
  4886.3  494.02  4912.9  492.66  4922.8  492.46  4939.6  491.23  4949.7  491.12
  4959.9  487.26  4968.0  482.80  4968.2  482.30  4971.7  482.30  4972.0  482.80
  4984.6  486.90  4990.2  489.55  4998.3  490.89  5003.3  490.89  5030.6  492.26
  5050.7  492.32  5065.5  491.75  5080.9  494.20  5101.0  495.52  5111.1  496.46
  5141.3  497.26  5172.5  498.56  5181.6  498.87  5191.6  499.79  5215.0  500.69
#Mann=6,-1,0
  4805.5    0.16       0  4886.3    0.12       0  4912.9    0.16       0
  4968.0    0.07       0  4972.0    0.16       0  5172.5    0.12       0
Bank Sta=4968,4972
Exp/Cntr=0.3,0.1

Type RM Length L Ch R = 1,36539,193,193,193
BEGIN DESCRIPTION:
Purtis Creek36538.82
END DESCRIPTION:
XS GIS Cut Line= 3
      2758887.92      6837741.24      2758794.59      6838014.28
      2758707.00      6838232.08
#Sta/Elev= 30
  4715.0  499.88  4746.5  498.60  4796.1  495.17  4858.7  493.43  4873.3  491.35
  4883.8  487.49  4890.0  487.30  4905.0  490.26  4916.5  490.94  4968.4  490.43
  4978.7  485.48  4983.7  484.90  4987.5  481.71  4987.8  481.21  4991.5  481.71
  4999.2  483.52  5003.6  483.52  5009.3  486.31  5014.7  487.05  5021.6  489.88
  5032.4  491.27  5068.4  490.91  5075.5  490.50  5086.2  488.03  5092.6  487.97
  5107.8  492.23  5146.4  497.36  5193.1  502.49  5205.5  504.11  5238.3  506.47
#Mann=5,-1,0
  4715.0    0.12       0  4916.5    0.16       0  4987.5    0.07       0
  4991.5    0.16       0  5193.1    0.12       0
Bank Sta=4987.5,4991.5
Exp/Cntr=0.3,0.1

Type RM Length L Ch R = 1,36346,228,228,228
BEGIN DESCRIPTION:
Purtis Creek36346.16
END DESCRIPTION:
XS GIS Cut Line= 3
      2758748.37      6837680.63      2758619.61      6837959.79
      2758536.02      6838134.39
#Sta/Elev= 30
  4691.5  500.24  4713.8  497.93  4724.9  497.57  4737.2  495.87  4769.0  493.84
  4813.0  492.60  4832.4  492.66  4857.5  492.64  4868.1  492.19  4903.4  488.84
  4927.2  488.65  4972.2  489.58  4978.2  487.98  4989.2  482.44  4995.3  481.01
  4995.5  480.51  4999.0  480.51  4999.3  481.01  5002.4  481.01  5011.3  486.23
  5017.9  489.06  5023.4  487.56  5033.5  488.32  5046.1  487.72  5068.7  488.54
  5108.5  495.26  5114.1  498.44  5144.4  504.06  5166.6  506.78  5192.5  507.73
#Mann=6,-1,0
  4691.5    0.05       0  4713.8    0.12       0  4832.4    0.16       0
  4927.2    0.12       0  4995.3    0.07       0  4999.3    0.12       0
Bank Sta=4995.3,4999.3
Exp/Cntr=0.3,0.1

Type RM Length L Ch R = 1,36118,167,167,167
BEGIN DESCRIPTION:
Purtis Creek36117.85
END DESCRIPTION:
XS GIS Cut Line= 3
      2758685.98      6837587.35      2758429.49      6837863.37
      2758337.67      6837966.40
#Sta/Elev= 30
  4622.6  499.00  4626.2  499.00  4632.2  497.57  4674.7  495.23  4688.8  493.74
  4772.6  492.35  4837.4  491.62  4879.9  488.95  4887.0  487.21  4915.1  487.18
  4936.6  488.90  4985.9  488.13  4993.3  486.42  4998.3  481.00  5007.5  481.44
  5012.2  479.66  5012.5  479.16  5016.2  479.66  5021.7  480.30  5028.4  485.90
  5033.5  487.20  5049.8  493.89  5056.9  497.65  5058.7  497.46  5063.6  496.95
  5071.1  499.66  5077.8  499.71  5085.3  502.43  5099.5  504.31  5137.4  505.54
#Mann=6,-1,0
  4622.6    0.05       0  4772.6    0.16       0  5012.2    0.07       0
  5016.2    0.16       0  5033.5    0.12       0  5058.7    0.16       0
Bank Sta=5012.2,5016.2
Exp/Cntr=0.3,0.1

Type RM Length L Ch R = 1,35951,139,139,139
BEGIN DESCRIPTION:
Purtis Creek35950.51
END DESCRIPTION:
XS GIS Cut Line= 3
      2758601.14      6837528.25      2758292.04      6837778.30
      2758200.48      6837864.31
#Sta/Elev= 30
  4602.7  496.75  4622.2  495.51  4636.2  493.68  4658.5  493.20  4679.3  491.44
  4737.9  489.25  4778.5  487.66  4821.6  484.88  4842.4  485.11  4867.7  487.17
  4885.6  488.13  4900.0  487.78  4928.7  484.75  4949.5  487.67  4970.4  487.67
  4984.7  486.87  4992.7  484.57  4996.5  479.63  4996.7  479.13  5000.2  479.13
  5000.5  479.63  5006.6  479.99  5013.5  481.55  5020.8  487.10  5027.6  490.48
  5034.9  497.95  5041.8  501.77  5049.1  502.81  5070.1  503.38  5125.9  503.47
#Mann=5,-1,0
  4602.7    0.05       0  4737.9    0.16       0  4867.7    0.12       0
  4996.5    0.07       0  5000.5    0.12       0
Bank Sta=4996.5,5000.5
Exp/Cntr=0.3,0.1

Type RM Length L Ch R = 1,35812,302,302,302
BEGIN DESCRIPTION:
Purtis Creek35812.08
END DESCRIPTION:
XS GIS Cut Line= 3
      2758562.57      6837453.69      2758273.23      6837645.79
      2758179.46      6837711.67
#Sta/Elev= 30
  4655.5  497.45  4658.5  496.73  4664.5  496.74  4715.7  493.13  4730.7  491.29
  4778.2  488.54  4795.4  488.65  4802.9  487.92  4817.9  487.93  4838.9  484.99
  4844.9  485.35  4854.0  484.69  4860.0  485.35  4896.1  485.39  4932.2  486.91
  4947.2  485.32  4953.3  483.10  4962.2  480.43  4966.2  478.25  4966.5  477.75
  4970.0  477.75  4970.2  478.25  4975.5  478.92  4983.3  482.71  4989.3  486.67
  4998.1  495.05  5011.6  501.30  5026.6  501.84  5075.8  502.05  5117.4  501.45
#Mann=6,-1,0
  4655.5    0.05       0  4778.2    0.12       0  4953.3    0.16       0
  4966.2    0.07       0  4970.2    0.16       0  5026.6    0.12       0
Bank Sta=4966.2,4970.2
Exp/Cntr=0.3,0.1

Type RM Length L Ch R = 1,35510,342,342,342
BEGIN DESCRIPTION:
Purtis Creek35510.13
END DESCRIPTION:
XS GIS Cut Line= 3
      2758415.04      6837202.59      2758301.58      6837411.97
      2758164.07      6837629.39
#Sta/Elev= 30
  4763.4  491.61  4784.3  490.38  4851.4  489.52  4857.0  488.69  4874.5  488.27
  4909.4  487.56  4938.8  488.20  4954.9  487.44  4960.7  484.11  4976.9  484.42
  4982.6  483.60  4989.1  480.09  4996.1  478.90  4996.4  478.40  4999.9  478.40
  5000.1  478.90  5001.5  478.90  5004.5  481.44  5007.1  482.47  5012.2  484.50
  5019.7  484.58  5062.1  481.96  5077.4  485.34  5096.6  485.12  5142.4  486.44
  5150.3  487.96  5165.6  489.21  5192.7  496.04  5223.2  500.43  5258.8  500.77
#Mann=6,-1,0
  4763.4    0.05       0  4874.5    0.16       0  4996.1    0.07       0
  5000.1    0.16       0  5007.1    0.12       0  5096.6    0.16       0
Bank Sta=4996.1,5000.1
Exp/Cntr=0.3,0.1

Type RM Length L Ch R = 1,35168,244,244,244
BEGIN DESCRIPTION:
Purtis Creek35168.14
END DESCRIPTION:
XS GIS Cut Line= 3
      2758362.37      6837103.87      2758165.56      6837265.78
      2758010.27      6837412.81
#Sta/Elev= 30
  4749.2  493.85  4794.8  490.48  4822.2  489.25  4836.4  487.73  4899.9  485.42
  4908.2  484.89  4914.6  483.66  4936.8  481.41  4943.3  483.17  4948.9  482.13
  4964.6  476.95  4970.0  474.53  4970.3  474.03  4973.8  474.03  4974.0  474.53
  4978.5  475.76  4986.4  481.33  5000.5  482.28  5007.3  482.10  5014.6  483.16
  5028.8  483.09  5042.9  484.78  5057.1  487.89  5064.0  488.68  5071.3  490.54
  5084.7  492.01  5106.5  493.74  5120.6  495.50  5134.8  496.34  5217.9  497.64
#Mann=6,-1,0
  4749.2    0.05       0  4899.9    0.12       0  4948.9    0.16       0
  4970.0    0.07       0  4974.0    0.16       0  5084.7    0.07       0
Bank Sta=4970,4974
Exp/Cntr=0.3,0.1

Type RM Length L Ch R = 1,34924,257,257,257
BEGIN DESCRIPTION:
Purtis Creek34924.48
END DESCRIPTION:
XS GIS Cut Line= 3
      2758278.27      6837013.07      2758048.74      6837085.42
      2757909.60      6837124.89
#Sta/Elev= 30
  4761.4  492.41  4784.8  492.00  4807.7  490.43  4840.0  489.63  4879.1  486.35
  4910.6  485.68  4924.9  484.56  4937.1  483.25  4942.4  483.49  4952.5  481.46
  4961.0  472.90  4961.2  472.40  4964.7  472.40  4965.0  472.90  4969.5  473.44
  4974.7  476.46  4984.0  479.15  5000.9  480.23  5025.7  480.91  5035.9  480.61
  5041.1  481.41  5067.3  478.67  5075.0  480.20  5080.2  481.96  5084.8  485.52
  5088.1  488.08  5098.5  491.01  5108.9  492.98  5114.1  494.76  5146.7  495.00
#Mann=5,-1,0
  4761.4    0.05       0  4924.9    0.12       0  4961.0    0.07       0
  4965.0    0.12       0  5084.8    0.16       0
Bank Sta=4961,4965
Exp/Cntr=0.3,0.1

Type RM Length L Ch R = 1,34667,212,212,212
BEGIN DESCRIPTION:
Purtis Creek34666.93
END DESCRIPTION:
XS GIS Cut Line= 3
      2758291.33      6836926.81      2757923.05      6836891.86
      2757799.59      6836886.71
#Sta/Elev= 30
  4632.6  492.15  4668.1  491.43  4688.2  489.55  4698.2  489.31  4718.3  487.23
  4738.4  486.36  4758.5  485.94  4768.5  486.32  4788.6  484.62  4818.8  484.40
  4858.9  481.84  4881.1  481.66  4929.3  480.33  4949.3  480.43  4961.6  478.43
  4967.4  473.57  4967.7  473.07  4971.2  473.07  4971.4  473.57  4979.5  474.73
  4989.5  477.45  5002.5  478.47  5009.6  480.21  5019.6  488.13  5029.6  491.34
  5036.4  492.12  5049.6  493.24  5089.7  492.97  5111.9  493.41  5126.1  493.45
#Mann=6,-1,0
  4632.6    0.05       0  4881.1    0.12       0  4967.4    0.07       0
  4971.4    0.12       0  5036.4    0.16       0  5111.9    0.07       0
Bank Sta=4967.4,4971.4
Exp/Cntr=0.3,0.1

Type RM Length L Ch R = 1,34455,155,155,155
BEGIN DESCRIPTION:
Purtis Creek34454.87
END DESCRIPTION:
XS GIS Cut Line= 3
      2758249.39      6836774.97      2758017.24      6836715.63
      2757844.80      6836678.54
#Sta/Elev= 30
  4762.3  489.29  4793.5  488.05  4835.9  486.57  4841.1  486.74  4869.0  484.52
  4900.0  483.49  4910.3  482.13  4917.6  479.95  4930.9  478.32  4958.4  476.63
  4963.6  474.36  4972.2  473.66  4982.6  473.85  4990.9  470.20  4991.1  469.70
  4994.6  469.70  4994.9  470.20  4999.2  473.13  5001.9  474.38  5005.1  474.38
  5013.4  476.89  5033.9  478.27  5043.4  476.38  5048.5  478.70  5064.6  480.33
  5074.8  482.70  5085.0  486.50  5092.7  487.81  5136.2  491.10  5178.3  491.86
#Mann=4,-1,0
  4762.3    0.12       0  4793.5    0.16       0  4990.9    0.07       0
  4994.9    0.16       0
Bank Sta=4990.9,4994.9
Exp/Cntr=0.3,0.1

Type RM Length L Ch R = 1,34300,129,129,129
BEGIN DESCRIPTION:
Purtis Creek34300.4
END DESCRIPTION:
XS GIS Cut Line= 3
      2758250.66      6836605.29      2757975.01      6836579.52
      2757800.72      6836570.09
#Sta/Elev= 30
  4724.0  485.23  4768.9  485.45  4824.0  482.72  4829.1  480.92  4849.2  478.62
  4859.2  478.42  4879.3  479.13  4909.5  477.05  4927.9  477.39  4932.9  476.77
  4939.6  477.24  4969.7  476.57  4979.8  474.84  4989.8  471.14  4995.8  469.59
  4996.1  469.09  4999.6  469.09  4999.8  469.59  5002.9  469.59  5009.9  475.41
  5019.9  476.16  5029.9  476.17  5039.9  484.29  5049.9  486.29  5065.5  487.61
  5100.0  488.43  5150.1  489.13  5160.1  488.62  5174.5  488.95  5175.4  489.02
#Mann=4,-1,0
  4724.0    0.16       0  4995.8    0.07       0  4999.8    0.16       0
  5174.5    0.07       0
Bank Sta=4995.8,4999.8
Exp/Cntr=0.3,0.1

Type RM Length L Ch R = 1,34171,181,181,181
BEGIN DESCRIPTION:
Purtis Creek34170.54
END DESCRIPTION:
XS GIS Cut Line= 3
      2758232.30      6836450.71      2758024.78      6836466.44
      2757823.33      6836473.65
#Sta/Elev= 30
  4790.9  483.32  4797.2  482.73  4817.3  481.59  4827.3  481.39  4867.4  481.71
  4927.6  480.14  4947.7  479.45  4957.7  478.39  4967.7  476.29  4977.7  470.26
  4985.8  470.22  4986.0  469.72  4989.5  469.72  4989.8  470.22  4993.0  472.09
  4999.0  472.31  5007.8  475.27  5017.8  476.44  5027.8  477.11  5037.8  478.87
  5047.8  482.01  5057.8  484.11  5077.8  484.78  5097.9  484.07  5117.9  483.96
  5137.9  484.41  5147.9  484.22  5177.9  484.74  5187.9  485.09  5200.6  485.13
#Mann=3,-1,0
  4790.9    0.16       0  4985.8    0.07       0  4989.8    0.16       0
Bank Sta=4985.8,4989.8
Exp/Cntr=0.3,0.1

Type RM Length L Ch R = 1,33990,218,218,218
BEGIN DESCRIPTION:
Purtis Creek33990.42
END DESCRIPTION:
XS GIS Cut Line= 3
      2758189.77      6836284.12      2758024.51      6836314.72
      2757872.57      6836366.20
#Sta/Elev= 30
  4833.9  479.93  4878.4  480.20  4896.4  479.50  4901.5  479.71  4908.9  478.55
  4919.1  477.68  4939.4  475.10  4954.4  475.58  4957.8  469.48  4958.0  468.98
  4961.5  468.98  4961.8  469.48  4969.9  471.94  4980.1  474.16  4990.3  474.78
  5002.0  474.61  5005.8  475.14  5011.1  474.93  5021.5  475.45  5032.0  474.74
  5037.2  475.13  5042.6  474.90  5053.2  476.96  5063.4  481.20  5068.7  481.56
  5094.8  481.49  5106.0  482.16  5126.2  482.29  5131.5  482.63  5162.4  482.53
#Mann=3,-1,0
  4833.9    0.16       0  4957.8    0.07       0  4961.8    0.16       0
Bank Sta=4957.8,4961.8
Exp/Cntr=0.3,0.1

Type RM Length L Ch R = 1,33772,206,206,206
BEGIN DESCRIPTION:
Purtis Creek33772.04
END DESCRIPTION:
XS GIS Cut Line= 3
      2757993.23      6836017.43      2757926.69      6836168.60
      2757841.07      6836346.17
#Sta/Elev= 30
  4839.6  476.24  4887.2  477.91  4902.5  476.98  4917.1  474.71  4922.5  474.52
  4940.4  475.44  4952.8  477.17  4963.7  476.18  4992.5  471.06  4998.0  473.47
  5003.3  471.74  5008.9  471.74  5015.4  468.38  5021.0  469.58  5027.6  466.58
  5027.9  466.08  5031.4  466.08  5031.6  466.58  5038.0  472.50  5043.6  470.00
  5051.8  474.14  5060.7  475.76  5066.2  475.91  5083.3  477.95  5096.2  480.03
  5118.4  481.60  5128.5  481.42  5151.1  482.12  5196.2  481.82  5201.9  481.34
#Mann=4,-1,0
  4839.6    0.12       0  4902.5    0.16       0  5027.6    0.07       0
  5031.6    0.16       0
Bank Sta=5027.6,5031.6
Exp/Cntr=0.3,0.1

Type RM Length L Ch R = 1,33566,188,188,188
BEGIN DESCRIPTION:
Purtis Creek33565.91
END DESCRIPTION:
XS GIS Cut Line= 3
      2757877.02      6835924.77      2757772.29      6836112.89
      2757685.23      6836277.36
#Sta/Elev= 30
  4788.4  475.52  4860.5  476.78  4866.2  476.42  4882.2  476.26  4925.6  477.21
  4969.1  476.15  4978.7  474.96  4985.1  467.22  4988.8  465.14  4989.1  464.64
  4992.6  464.64  4992.8  465.14  5003.7  465.54  5006.8  470.29  5012.9  472.66
  5023.2  473.18  5035.5  472.20  5050.9  472.59  5058.1  473.99  5066.9  477.94
  5072.9  476.62  5080.8  478.96  5089.2  479.59  5094.9  478.59  5103.4  478.97
  5116.9  478.84  5126.0  477.90  5138.9  477.54  5148.7  477.53  5189.8  479.02
#Mann=4,-1,0
  4788.4    0.16       0  4988.8    0.07       0  4992.8    0.16       0
  5066.9    0.07       0
Bank Sta=4988.8,4992.8
Exp/Cntr=0.3,0.1

Type RM Length L Ch R = 1,33378,94,94,94
BEGIN DESCRIPTION:
Purtis Creek33378.46
END DESCRIPTION:
XS GIS Cut Line= 3
      2757816.57      6835852.56      2757728.84      6835966.36
      2757565.32      6836225.60
#Sta/Elev= 30
  4858.5  475.91  4944.1  475.18  4950.4  473.91  4964.9  473.26  4971.2  471.11
  4979.4  471.33  4985.7  468.83  4991.9  464.28  4992.1  463.78  4995.6  463.78
  4995.9  464.28  5000.2  468.75  5015.2  471.13  5021.2  471.16  5036.4  472.57
  5051.7  472.06  5057.6  472.63  5066.8  472.15  5072.9  470.62  5078.8  470.05
  5088.2  471.09  5094.1  470.85  5099.0  471.60  5109.4  472.26  5115.3  471.48
  5137.7  471.08  5161.2  475.39  5182.3  476.56  5224.7  475.92  5308.7  477.03
#Mann=4,-1,0
  4858.5    0.16       0  4991.9    0.07       0  4995.9    0.16       0
  5099.0    0.07       0
Bank Sta=4991.9,4995.9
Exp/Cntr=0.3,0.1

Type RM Length L Ch R = 1,33284,167,167,167
BEGIN DESCRIPTION:
Purtis Creek33284.04
END DESCRIPTION:
XS GIS Cut Line= 3
      2757772.97      6835845.79      2757663.72      6835897.68
      2757380.91      6836173.08
#Sta/Elev= 30
  4878.3  475.76  4886.0  476.07  4919.2  475.66  4925.1  474.88  4930.6  475.33
  4947.8  473.94  4953.3  474.41  4970.5  473.98  4993.3  471.35  4997.3  470.33
  5014.1  470.69  5021.3  469.68  5028.2  463.93  5033.4  463.23  5033.7  462.73
  5037.2  462.73  5037.4  463.23  5042.4  469.31  5049.5  471.87  5061.6  474.04
  5063.7  474.47  5084.8  475.38  5134.4  474.50  5198.0  474.92  5233.4  474.31
  5261.6  475.10  5284.8  475.26  5318.1  475.68  5367.7  476.96  5394.0  476.62
#Mann=5,-1,0
  4878.3    0.16       0  5033.4    0.07       0  5037.4    0.16       0
  5061.6    0.07       0  5284.8    0.05       0
Bank Sta=5033.4,5037.4
Exp/Cntr=0.3,0.1

Type RM Length L Ch R = 1,33117,206,206,206
BEGIN DESCRIPTION:
Purtis Creek33116.74
END DESCRIPTION:
XS GIS Cut Line= 3
      2757701.30      6835620.66      2757568.83      6835766.78
      2757273.49      6836116.80
#Sta/Elev= 30
  4804.2  483.58  4872.1  482.58  4893.2  480.59  4899.9  480.86  4914.1  479.91
  4921.6  478.75  4928.3  478.66  4942.5  476.73  4950.0  474.53  4956.7  471.11
  4964.1  468.56  4985.1  469.14  4992.5  468.36  5001.4  464.54  5007.5  464.54
  5011.3  463.58  5011.6  463.08  5015.4  463.08  5015.7  463.58  5020.1  466.22
  5027.8  467.43  5031.4  470.33  5034.4  472.75  5055.4  472.33  5091.5  474.33
  5155.3  473.20  5248.5  473.40  5304.8  474.34  5325.6  474.01  5459.4  476.16
#Mann=6,-1,0
  4804.2    0.12       0  5011.3    0.07       0  5015.7    0.12       0
  5031.4    0.16       0  5055.4    0.07       0  5248.5    0.05       0
Bank Sta=5011.3,5015.7
Exp/Cntr=0.3,0.1

Type RM Length L Ch R = 1,32911,172,172,172
BEGIN DESCRIPTION:
Purtis Creek32911.41
END DESCRIPTION:
XS GIS Cut Line= 3
      2757651.57      6835613.36      2757418.05      6835668.29
      2757057.04      6835836.09
#Sta/Elev= 30
  4765.4  481.67  4819.0  478.71  4832.8  478.49  4861.4  476.03  4866.5  476.17
  4884.1  474.08  4903.7  472.71  4935.5  471.49  4966.3  471.75  4976.6  469.95
  4986.9  469.10  5009.2  468.66  5018.3  466.70  5023.8  466.73  5027.3  461.51
  5027.7  461.01  5031.6  461.01  5031.9  461.51  5040.6  463.32  5046.7  468.79
  5069.6  468.00  5084.7  468.39  5092.5  471.68  5098.0  471.45  5106.8  473.33
  5126.8  472.81  5150.9  472.09  5189.6  472.08  5249.7  473.10  5403.4  475.71
#Mann=6,-1,0
  4765.4    0.12       0  4866.5    0.16       0  5027.3    0.07       0
  5031.9    0.16       0  5126.8    0.07       0  5249.7    0.05       0
Bank Sta=5027.3,5031.9
Exp/Cntr=0.3,0.1
