--- Purtis Creek Trib C.prj (project) ---

Proj Title=Purtis Creek Trib C Base Level Engineering
Current Plan=p01
Default Exp/Contr=0.3,0.1
English Units
Geom File=g01
Flow File=f01
Plan File=p01
BEGIN DESCRIPTION:
Purtis Creek Trib C
END DESCRIPTION:

--- Purtis Creek Trib C.p01 (plan) ---

Plan Title=Multiple Run
Short Identifier=Multiple
Geom File=g01
Flow File=f01
Subcritical Flow
K Sum by GR= 0
Std Step Tol= 0.01
Critical Tol= 0.01
Num of Std Step Trials= 20
Max Error Tol= 0.3
Flow Tol Ratio= 0.001
Split Flow NTrial= 30
Split Flow Tol= 0.02
Split Flow Ratio= 0.02
Log Output Level= 0
Friction Slope Method= 1
Unsteady Friction Slope Method= 2
Unsteady Bridges Friction Slope Method= 1
Parabolic Critical Depth
Global Vel Dist=  1 , 1 , 1
Global Log Level= 0
CheckData=True
Encroach Param= -1, 0, 0, 0
BEGIN DESCRIPTION:
Multiple Run
END DESCRIPTION:

--- Purtis Creek Trib C.f01 (steady flow) ---

Flow Title=Multiple
Number of Profiles=7
Profile Names=10-year,25-year,50-year,1pct_min,100-year,1pct_plu,500-year
River Rch & RM= Purtis Creek Tri,Reach-1,8218
     528     712     863     521    1040    2074    1510
River Rch & RM= Purtis Creek Tri,Reach-1,2534
     650     886    1081     656    1309    2611    1923
Boundary for River Rch & Prof#=Purtis Creek Tri,Reach-1,1
Up Type=0
Dn Type=3
Dn Slope=0.005
Boundary for River Rch & Prof#=Purtis Creek Tri,Reach-1,2
Up Type=0
Dn Type=3
Dn Slope=0.005
Boundary for River Rch & Prof#=Purtis Creek Tri,Reach-1,3
Up Type=0
Dn Type=3
Dn Slope=0.005
Boundary for River Rch & Prof#=Purtis Creek Tri,Reach-1,4
Up Type=0
Dn Type=3
Dn Slope=0.005
Boundary for River Rch & Prof#=Purtis Creek Tri,Reach-1,5
Up Type=0
Dn Type=3
Dn Slope=0.005
Boundary for River Rch & Prof#=Purtis Creek Tri,Reach-1,6
Up Type=0
Dn Type=3
Dn Slope=0.005
Boundary for River Rch & Prof#=Purtis Creek Tri,Reach-1,7
Up Type=0
Dn Type=3
Dn Slope=0.005

--- Purtis Creek Trib C.g01 (geometry) ---

Geom Title=Existing Conditions

River Reach=Purtis Creek Tri,Reach-1
Reach XY= 30
      2756076.00      6831811.00      2755928.71      6831566.40
      2755277.55      6831457.25      2755137.11      6831371.32
      2755082.80      6831118.86      2754584.32      6830957.84
      2754517.82      6830813.83      2754422.68      6830852.94
      2754278.66      6830716.46      2753815.94      6830550.39
      2753762.80      6830297.27      2753431.28      6830105.46
      2753370.98      6829866.02      2753233.72      6829857.83
      2753069.96      6829662.62      2752875.92      6829753.70
      2752446.03      6829611.06      2752240.04      6829710.91
      2752026.00      6829461.00      2751825.91      6829553.70
      2751696.37      6829460.62      2751524.37      6829657.87
      2751237.03      6829562.27      2751182.52      6829703.32
      2750987.83      6829712.65      2750770.02      6829858.84
      2750420.93      6829760.16      2750279.41      6829903.56
      2750211.30      6829811.31      2750126.00      6829861.00

Type RM Length L Ch R = 1,8218,145,145,145
BEGIN DESCRIPTION:
Purtis Creek Trib C8217.94
END DESCRIPTION:
XS GIS Cut Line= 3
      2756183.74      6831573.41      2756061.07      6831796.17
      2755974.94      6832001.32
#Sta/Elev= 30
  4745.7  471.03  4750.0  470.52  4777.5  469.05  4831.4  467.37  4858.9  464.68
  4875.0  464.52  4880.7  463.95  4891.1  464.27  4896.8  463.61  4912.9  463.79
  4918.6  463.42  4925.6  463.59  4940.3  463.18  4956.4  463.59  4971.3  463.39
  4976.2  462.79  4976.4  462.29  4979.9  462.29  4980.2  462.79  5016.1  463.06
  5029.2  463.66  5052.9  463.16  5100.5  463.64  5153.4  464.79  5167.9  465.28
  5177.2  466.00  5182.6  467.47  5189.6  468.31  5206.4  469.24  5222.5  469.59
#Mann=3,-1,0
  4745.7    0.05       0  4976.2    0.05       0  4980.2    0.05       0
Bank Sta=4976.2,4980.2
Exp/Cntr=0.3,0.1

Type RM Length L Ch R = 1,8073,147,147,147
BEGIN DESCRIPTION:
Purtis Creek Trib C8072.71
END DESCRIPTION:
XS GIS Cut Line= 3
      2756099.44      6831478.16      2755974.23      6831686.84
      2755862.13      6831899.77
#Sta/Elev= 30
  4759.9  468.84  4778.5  468.42  4794.1  468.44  4799.9  467.68  4809.6  467.72
  4821.5  466.83  4831.0  466.78  4844.8  465.93  4858.2  465.48  4867.9  463.42
  4873.7  463.01  4879.8  462.05  4926.2  462.37  4936.1  461.90  4936.4  461.40
  4939.9  461.40  4940.1  461.90  4947.6  462.56  4953.4  462.23  4996.5  462.55
  5028.3  462.44  5033.9  462.15  5050.3  463.14  5056.0  463.06  5100.0  465.44
  5166.2  468.14  5198.9  468.91  5211.4  468.77  5226.6  469.20  5243.9  469.21
#Mann=3,-1,0
  4759.9    0.05       0  4936.1    0.05       0  4940.1    0.05       0
Bank Sta=4936.1,4940.1
Exp/Cntr=0.3,0.1

Type RM Length L Ch R = 1,7926,96,96,96
BEGIN DESCRIPTION:
Purtis Creek Trib C7926.09
END DESCRIPTION:
XS GIS Cut Line= 3
      2755974.43      6831406.31      2755918.82      6831563.40
      2755826.39      6831829.99
#Sta/Elev= 30
  4834.0  467.68  4839.1  467.68  4860.2  466.06  4869.9  465.96  4875.2  465.52
  4892.0  465.01  4906.1  464.98  4945.1  463.28  4962.6  462.93  4987.5  461.92
  5000.6  462.00  5006.7  461.62  5006.9  461.12  5010.4  461.12  5010.7  461.62
  5072.2  462.49  5081.5  462.26  5086.8  462.62  5093.4  462.31  5103.9  462.38
  5118.0  462.89  5125.1  463.58  5135.7  463.74  5188.6  467.14  5206.1  467.66
  5237.2  467.58  5242.5  468.06  5262.7  467.57  5268.4  467.92  5282.8  467.92
#Mann=3,-1,0
  4834.0    0.05       0  5006.7    0.05       0  5010.7    0.05       0
Bank Sta=5006.7,5010.7
Exp/Cntr=0.3,0.1

Type RM Length L Ch R = 1,7830,104,104,104
BEGIN DESCRIPTION:
Purtis Creek Trib C7829.75
END DESCRIPTION:
XS GIS Cut Line= 3
      2755879.11      6831383.20      2755823.08      6831557.18
      2755751.49      6831782.71
#Sta/Elev= 30
  4819.3  466.70  4838.0  465.68  4849.8  465.76  4869.5  463.74  4901.0  462.37
  4922.0  461.83  4932.6  461.95  4946.0  461.29  4953.6  461.52  4985.1  460.91
  4995.6  460.95  5001.5  461.64  5005.5  461.64  5014.6  460.81  5014.8  460.31
  5018.3  460.31  5018.6  460.81  5037.2  461.60  5069.0  461.37  5079.9  462.11
  5100.5  462.75  5106.9  463.59  5132.0  464.87  5139.2  465.73  5163.5  465.72
  5171.5  466.12  5176.7  465.73  5203.7  466.56  5215.9  466.18  5238.7  466.24
#Mann=3,-1,0
  4819.3    0.05       0  5014.6    0.05       0  5018.6    0.05       0
Bank Sta=5014.6,5018.6
Exp/Cntr=0.3,0.1

Type RM Length L Ch R = 1,7726,113,113,113
BEGIN DESCRIPTION:
Purtis Creek Trib C7726.03
END DESCRIPTION:
XS GIS Cut Line= 3
      2755763.17      6831346.61      2755734.90      6831512.18
      2755691.41      6831767.13
#Sta/Elev= 30
  4833.6  465.83  4849.9  465.38  4868.5  465.76  4878.6  464.14  4888.8  464.94
  4898.9  464.21  4905.0  463.15  4919.2  462.62  4939.5  462.24  4965.1  460.87
  4990.2  460.57  4998.4  461.06  5001.6  461.06  5010.5  460.78  5025.2  460.86
  5039.0  460.48  5039.2  459.98  5042.7  459.98  5043.0  460.48  5051.1  461.18
  5080.3  461.00  5091.7  462.22  5101.8  462.52  5132.3  462.91  5140.5  463.25
  5145.6  463.11  5200.7  464.33  5205.7  464.07  5213.4  464.40  5260.2  465.26
#Mann=3,-1,0
  4833.6    0.05       0  5039.0    0.05       0  5043.0    0.05       0
Bank Sta=5039,5043
Exp/Cntr=0.3,0.1

Type RM Length L Ch R = 1,7613,422,422,422
BEGIN DESCRIPTION:
Purtis Creek Trib C7612.78
END DESCRIPTION:
XS GIS Cut Line= 3
      2755644.83      6831317.77      2755622.58      6831508.15
      2755592.20      6831760.65
#Sta/Elev= 30
  4811.7  465.21  4842.4  464.99  4865.3  465.42  4875.4  464.81  4885.4  463.29
  4905.6  463.36  4930.8  461.60  4935.8  461.82  4962.3  460.10  4966.0  459.90
  4986.1  460.26  5000.3  459.65  5000.5  459.15  5004.0  459.15  5004.3  459.65
  5007.3  459.65  5013.9  460.61  5023.3  460.61  5046.5  460.35  5076.8  462.09
  5086.8  462.49  5101.1  462.32  5127.1  463.50  5137.2  463.58  5147.3  464.42
  5157.3  464.31  5183.3  465.22  5188.3  465.00  5217.8  465.75  5257.7  466.16
#Mann=5,-1,0
  4811.7    0.05       0  4962.3    0.16       0  5000.3    0.07       0
  5004.3    0.16       0  5023.3    0.05       0
Bank Sta=5000.3,5004.3
Exp/Cntr=0.3,0.1

Type RM Length L Ch R = 1,7191,138,138,138
BEGIN DESCRIPTION:
Purtis Creek Trib C7190.81
END DESCRIPTION:
XS GIS Cut Line= 5
      2755624.93      6831356.07      2755580.07      6831425.67
      2755250.81      6831413.78      2755226.42      6831419.68
      2754970.16      6831429.01
#Sta/Elev= 30
  4566.9  465.34  4584.7  465.79  4591.6  464.34  4606.8  463.18  4620.4  463.05
  4627.9  463.80  4643.1  463.00  4654.2  463.36  4693.8  461.03  4753.8  460.22
  4773.9  460.86  4793.9  459.18  4813.9  459.22  4823.9  459.99  4873.9  458.96
  4913.3  459.02  4924.0  459.73  4944.0  459.47  4964.0  458.37  4988.9  458.50
  4994.4  457.81  5042.2  456.99  5064.7  457.63  5102.8  456.51  5103.0  456.01
  5106.5  456.01  5106.8  456.51  5173.9  460.52  5234.8  460.37  5260.7  461.68
#Mann=5,-1,0
  4566.9    0.05       0  4620.4    0.16       0  5042.2    0.05       0
  5102.8    0.07       0  5106.8    0.05       0
Bank Sta=5102.8,5106.8
Exp/Cntr=0.3,0.1

Type RM Length L Ch R = 1,7053,91,91,91
BEGIN DESCRIPTION:
Purtis Creek Trib C7053.2
END DESCRIPTION:
XS GIS Cut Line= 3
      2755555.43      6831352.33      2755141.13      6831346.18
      2754930.83      6831341.07
#Sta/Elev= 30
  4586.1  465.05  4605.5  464.93  4615.5  464.47  4675.5  464.33  4705.5  463.66
  4715.5  464.06  4725.5  462.66  4745.5  463.16  4805.6  461.86  4815.6  461.93
  4835.6  460.57  4855.6  459.70  4915.6  459.08  4935.6  458.16  4945.6  457.35
  4985.6  457.36  5000.4  457.02  5013.6  454.87  5013.8  454.37  5017.3  454.37
  5017.6  454.87  5035.6  456.93  5055.6  456.09  5075.6  457.19  5085.6  457.44
  5115.6  457.05  5125.6  457.32  5145.6  458.75  5165.6  459.60  5210.8  460.31
#Mann=3,-1,0
  4586.1    0.05       0  5013.6    0.05       0  5017.6    0.05       0
Bank Sta=5013.6,5017.6
Exp/Cntr=0.3,0.1

Type RM Length L Ch R = 1,6962,84,84,84
BEGIN DESCRIPTION:
Purtis Creek Trib C6962.16
END DESCRIPTION:
XS GIS Cut Line= 3
      2755298.73      6831236.14      2755139.52      6831275.55
      2754941.59      6831329.65
#Sta/Elev= 30
  4837.3  461.98  4850.4  461.70  4871.0  460.82  4877.2  460.34  4891.6  459.60
  4912.2  458.97  4918.7  458.35  4943.1  457.78  4953.4  457.71  4958.1  453.47
  4958.3  452.97  4961.8  452.97  4962.1  453.47  4965.2  454.51  4974.0  456.32
  4994.6  455.77  5006.6  455.94  5046.4  455.72  5075.6  455.75  5080.8  455.05
  5087.9  455.82  5098.3  455.82  5108.6  456.12  5115.3  456.66  5120.5  456.62
  5149.8  458.36  5160.5  458.80  5189.5  459.15  5194.7  459.71  5206.5  459.76
#Mann=3,-1,0
  4837.3    0.05       0  4958.1    0.05       0  4962.1    0.05       0
Bank Sta=4958.1,4962.1
Exp/Cntr=0.3,0.1

Type RM Length L Ch R = 1,6878,170,170,170
BEGIN DESCRIPTION:
Mapping XS b0eedcee
END DESCRIPTION:
XS GIS Cut Line= 3
      2755231.69      6831123.67      2755081.75      6831215.29
      2754941.05      6831321.83
#Sta/Elev= 30
  4826.9  461.84  4835.4  461.05  4857.0  459.68  4866.3  459.40  4915.6  457.06
  4924.4  456.43  4939.0  455.86  4945.7  455.20  4951.5  455.25  4961.1  454.78
  4974.2  454.81  4982.4  452.12  4986.3  452.09  4986.5  451.59  4990.0  451.59
  4990.3  452.09  4997.2  455.51  5018.2  455.71  5039.1  455.62  5047.3  456.37
  5053.6  456.33  5060.0  456.79  5068.2  457.08  5089.0  457.19  5110.2  457.69
  5118.1  457.65  5124.4  457.94  5132.7  457.89  5138.9  458.28  5179.1  459.34
#Mann=3,-1,0
  4826.9    0.05       0  4986.3    0.05       0  4990.3    0.05       0
Bank Sta=4986.3,4990.3
Exp/Cntr=0.3,0.1

Type RM Length L Ch R = 1,6708,103,103,103
BEGIN DESCRIPTION:
Purtis Creek Trib C6744.73
END DESCRIPTION:
XS GIS Cut Line= 4
      2755093.85      6830928.94      2755035.25      6831110.83
      2754974.98      6831255.13      2754930.14      6831328.31
#Sta/Elev= 30
  4808.9  461.41  4812.6  461.41  4817.3  460.88  4874.1  460.41  4881.4  460.19
  4886.6  459.43  4895.1  458.90  4913.5  456.85  4918.7  455.85  4926.6  453.84
  4935.1  449.31  4935.4  448.81  4938.9  448.81  4939.1  449.31  4944.0  451.03
  4950.8  453.12  4958.1  454.21  4968.7  454.00  4977.6  452.24  4982.8  452.12
  4989.7  453.33  5003.8  453.85  5037.5  455.43  5085.2  455.78  5090.6  455.40
  5114.4  456.13  5119.8  455.89  5143.6  456.28  5203.3  458.31  5242.2  460.09
#Mann=5,-1,0
  4808.9    0.05       0  4935.1    0.07       0  4939.1    0.05       0
  4944.0    0.16       0  5003.8    0.05       0
Bank Sta=4935.1,4939.1
Exp/Cntr=0.3,0.1

Type RM Length L Ch R = 1,6605,93,93,93
BEGIN DESCRIPTION:
Purtis Creek Trib C6604.63
END DESCRIPTION:
XS GIS Cut Line= 3
      2754951.56      6830883.53      2754943.06      6831082.45
      2754940.26      6831273.92
#Sta/Elev= 30
  4804.8  461.99  4817.6  460.98  4822.6  460.92  4842.3  459.29  4852.3  459.16
  4908.7  457.56  4932.4  456.08  4962.4  455.10  4972.4  454.55  4982.4  450.91
  4990.4  449.82  4990.7  449.32  4994.2  449.32  4994.4  449.82  5000.7  453.45
  5003.9  453.45  5012.5  452.10  5042.5  454.05  5047.1  453.98  5052.5  453.90
  5062.5  454.17  5082.5  454.11  5092.5  454.29  5122.5  455.30  5141.1  456.75
  5146.1  456.65  5152.5  457.26  5182.5  457.67  5191.5  458.05  5195.4  458.05
#Mann=5,-1,0
  4804.8    0.05       0  4908.7    0.16       0  4990.4    0.07       0
  4994.4    0.16       0  5047.1    0.05       0
Bank Sta=4990.4,4994.4
Exp/Cntr=0.3,0.1

Type RM Length L Ch R = 1,6512,83,83,83
BEGIN DESCRIPTION:
Purtis Creek Trib C6511.88
END DESCRIPTION:
XS GIS Cut Line= 3
      2754864.31      6830883.49      2754855.34      6831064.08
      2754846.84      6831262.99
#Sta/Elev= 30
  4822.2  457.91  4849.7  457.01  4869.8  456.77  4886.8  456.15  4889.2  456.63
  4891.8  457.15  4899.8  456.44  4929.8  455.39  4939.9  454.46  4959.9  454.08
  4979.9  452.89  4989.9  451.77  4997.0  448.36  4997.2  447.86  5000.7  447.86
  5001.0  448.36  5003.0  448.36  5009.9  451.84  5019.9  452.77  5040.0  453.16
  5070.0  454.21  5075.8  454.52  5090.0  455.22  5104.8  455.47  5120.0  456.43
  5140.1  457.18  5150.1  457.71  5180.1  458.73  5198.6  459.82  5202.1  459.82
#Mann=5,-1,0
  4822.2   0.035       0  4889.2    0.16       0  4997.0    0.07       0
  5001.0    0.16       0  5075.8    0.05       0
Bank Sta=4997,5001
Exp/Cntr=0.3,0.1

Type RM Length L Ch R = 1,6429,83,83,83
BEGIN DESCRIPTION:
Purtis Creek Trib C6428.73
END DESCRIPTION:
XS GIS Cut Line= 4
      2754866.43      6830833.81      2754784.66      6831024.49
      2754751.50      6831103.78      2754704.33      6831192.51
#Sta/Elev= 30
  4795.0  459.45  4802.8  459.20  4808.5  458.68  4814.0  461.18  4832.1  460.24
  4837.5  458.96  4855.7  458.46  4861.1  457.55  4879.0  456.70  4884.7  456.82
  4890.1  456.23  4920.7  455.06  4944.3  454.62  4955.2  454.81  4966.2  453.85
  4982.0  452.95  4989.8  452.28  4997.9  451.14  5002.5  451.14  5006.0  447.81
  5006.3  447.31  5009.8  447.31  5010.0  447.81  5013.4  447.84  5020.4  449.10
  5031.2  451.84  5037.2  452.31  5052.9  452.44  5096.6  455.00  5188.9  459.52
#Mann=5,-1,0
  4795.0   0.035       0  4920.7    0.16       0  4982.0   0.035       0
  5006.0   0.035       0  5010.0   0.035       0
Bank Sta=5006,5010
Exp/Cntr=0.3,0.1

Type RM Length L Ch R = 1,6346,140,140,140
BEGIN DESCRIPTION:
Purtis Creek Trib C6345.64
END DESCRIPTION:
XS GIS Cut Line= 4
      2754802.84      6830766.27      2754708.15      6830997.74
      2754657.27      6831088.50      2754598.51      6831166.01
#Sta/Elev= 30
  4753.9  462.09  4766.4  461.82  4877.9  456.03  4949.5  453.22  4964.3  451.98
  4969.9  448.60  4975.3  451.66  4985.9  447.40  4991.9  446.52  4992.1  446.02
  4995.6  446.02  4995.9  446.52  5016.0  446.91  5030.7  449.12  5034.4  450.16
  5037.7  451.09  5043.5  451.68  5053.2  451.79  5059.4  452.25  5081.1  452.12
  5097.1  453.16  5102.8  452.76  5106.6  453.75  5147.0  454.95  5153.3  455.99
  5167.9  456.37  5174.1  457.62  5182.4  457.64  5188.7  459.39  5205.3  460.86
#Mann=7,-1,0
  4753.9   0.035       0  4766.4    0.05       0  4949.5   0.035       0
  4991.9   0.035       0  4995.9   0.035       0  5034.4    0.07       0
  5053.2    0.05       0
Bank Sta=4991.9,4995.9
Exp/Cntr=0.3,0.1

Type RM Length L Ch R = 1,6206,164,164,164
BEGIN DESCRIPTION:
Purtis Creek Trib C6205.92
END DESCRIPTION:
XS GIS Cut Line= 3
      2754688.34      6830736.34      2754581.59      6830957.14
      2754510.91      6831102.07
#Sta/Elev= 30
  4755.8  458.61  4769.6  458.34  4783.2  457.14  4826.4  455.33  4860.0  453.78
  4865.5  453.14  4933.3  450.90  4938.9  449.93  4949.8  449.17  4955.9  449.68
  4961.5  447.68  4972.0  447.90  4978.5  446.98  4992.2  443.24  4992.5  442.74
  4996.0  442.74  4996.2  443.24  5006.7  446.92  5016.5  448.79  5023.6  450.49
  5037.7  450.54  5046.2  451.26  5051.7  452.30  5061.0  455.49  5068.7  457.05
  5074.3  457.49  5119.3  459.40  5136.3  459.56  5141.8  460.01  5162.3  460.00
#Mann=5,-1,0
  4755.8    0.05       0  4826.4    0.07       0  4992.2    0.07       0
  4996.2    0.07       0  5037.7    0.05       0
Bank Sta=4992.2,4996.2
Exp/Cntr=0.3,0.1

Type RM Length L Ch R = 1,6042,155,155,155
BEGIN DESCRIPTION:
Purtis Creek Trib C6042.12
END DESCRIPTION:
XS GIS Cut Line= 3
      2754540.84      6830683.39      2754514.40      6830819.14
      2754469.23      6831045.37
#Sta/Elev= 30
  4868.1  457.42  4886.0  456.31  4920.6  455.06  4937.0  453.48  4947.2  451.67
  4967.2  449.66  4972.3  447.17  4977.7  443.49  4987.9  447.03  4998.1  448.41
  5002.8  442.65  5003.0  442.15  5006.5  442.15  5006.8  442.65  5009.9  442.65
  5023.7  444.98  5028.8  444.52  5038.9  449.24  5049.1  450.33  5059.3  450.47
  5079.8  452.24  5110.3  453.54  5120.5  454.22  5146.6  455.01  5161.3  456.20
  5176.8  456.63  5191.8  456.69  5212.2  457.33  5227.8  458.54  5237.1  458.31
#Mann=4,-1,0
  4868.1    0.07       0  5002.8    0.07       0  5006.8    0.07       0
  5146.6    0.05       0
Bank Sta=5002.8,5006.8
Exp/Cntr=0.3,0.1

Type RM Length L Ch R = 1,5887,162,162,162
BEGIN DESCRIPTION:
Purtis Creek Trib C5886.59
END DESCRIPTION:
XS GIS Cut Line= 3
      2754413.12      6830632.27      2754385.30      6830825.10
      2754365.40      6831056.52
#Sta/Elev= 30
  4807.5  456.85  4821.8  457.08  4826.9  456.28  4844.7  456.01  4876.9  454.75
  4897.3  454.40  4927.5  452.75  4937.6  450.70  4947.7  449.70  4957.6  449.18
  4962.6  448.61  5008.2  448.44  5018.3  447.51  5026.3  442.83  5026.6  442.33
  5030.1  442.33  5030.3  442.83  5038.4  447.64  5047.9  449.03  5058.4  450.16
  5068.5  450.69  5087.7  451.16  5138.7  453.73  5148.8  455.04  5171.5  454.80
  5178.9  456.18  5188.9  455.90  5198.9  455.99  5229.1  457.33  5234.6  457.94
#Mann=5,-1,0
  4807.5    0.05       0  4844.7    0.07       0  5026.3    0.07       0
  5030.3    0.07       0  5087.7    0.05       0
Bank Sta=5026.3,5030.3
Exp/Cntr=0.3,0.1

Type RM Length L Ch R = 1,5725,107,107,107
BEGIN DESCRIPTION:
Purtis Creek Trib C5724.85
END DESCRIPTION:
XS GIS Cut Line= 3
      2754306.34      6830536.10      2754282.01      6830721.28
      2754261.15      6830945.44
#Sta/Elev= 30
  4815.8  455.48  4851.0  454.63  4861.5  454.01  4911.5  452.41  4930.1  451.51
  4941.8  450.70  4951.9  449.66  4961.9  443.56  4972.0  441.12  4982.1  441.29
  4988.0  440.98  4990.2  440.87  4990.5  440.37  4994.0  440.37  4994.2  440.87
  4999.9  441.83  5004.9  441.83  5010.4  444.11  5015.4  443.34  5022.4  445.58
  5033.8  446.80  5062.6  447.71  5072.6  448.22  5132.9  452.15  5152.9  452.62
  5173.0  453.46  5183.1  453.94  5193.1  454.75  5213.2  455.92  5227.7  456.26
#Mann=5,-1,0
  4815.8    0.05       0  4988.0    0.07       0  4990.2    0.07       0
  4994.2    0.07       0  5033.8    0.05       0
Bank Sta=4990.2,4994.2
Exp/Cntr=0.3,0.1

Type RM Length L Ch R = 1,5618,141,141,141
BEGIN DESCRIPTION:
Purtis Creek Trib C5618.32
END DESCRIPTION:
XS GIS Cut Line= 3
      2754197.53      6830477.67      2754177.61      6830708.36
      2754171.73      6830905.62
#Sta/Elev= 30
  4769.6  454.97  4773.8  454.97  4803.1  453.85  4813.1  453.74  4841.9  452.53
  4846.9  451.98  4853.2  451.66  4903.4  450.65  4923.5  449.49  4953.6  448.66
  4960.2  448.31  4965.2  447.64  4973.7  447.41  4983.7  446.90  4991.8  441.23
  4992.0  440.73  4995.5  440.73  4995.8  441.23  5000.0  441.48  5005.0  441.48
  5013.8  447.62  5023.8  448.71  5043.8  449.46  5073.8  451.97  5083.8  452.53
  5113.8  453.52  5143.9  454.07  5183.9  455.87  5193.7  456.26  5198.5  456.26
#Mann=3,-1,0
  4769.6    0.05       0  4991.8    0.05       0  4995.8    0.05       0
Bank Sta=4991.8,4995.8
Exp/Cntr=0.3,0.1

Type RM Length L Ch R = 1,5477,132,132,132
BEGIN DESCRIPTION:
Purtis Creek Trib C5476.84
END DESCRIPTION:
XS GIS Cut Line= 3
      2754081.19      6830484.23      2754056.29      6830647.30
      2754017.84      6830915.19
#Sta/Elev= 30
  4840.7  455.98  4848.2  454.98  4877.9  452.78  4898.1  451.86  4905.7  450.51
  4910.8  450.77  4918.4  450.05  4949.4  448.33  4958.8  448.00  4968.9  446.86
  4979.3  446.43  4989.2  444.81  5003.0  439.41  5003.3  438.91  5006.8  438.91
  5007.0  439.41  5010.1  439.41  5019.5  441.88  5029.6  448.12  5038.8  448.61
  5059.9  448.14  5109.3  449.16  5114.4  448.85  5160.9  450.15  5179.9  451.09
  5184.9  450.95  5241.8  453.91  5250.4  454.17  5255.5  453.85  5276.3  454.51
#Mann=5,-1,0
  4840.7    0.05       0  4848.2    0.16       0  4949.4    0.05       0
  5003.0    0.05       0  5007.0    0.05       0
Bank Sta=5003,5007
Exp/Cntr=0.3,0.1

Type RM Length L Ch R = 1,5345,159,159,159
BEGIN DESCRIPTION:
Purtis Creek Trib C5344.8
END DESCRIPTION:
XS GIS Cut Line= 3
      2754002.11      6830426.51      2753933.64      6830614.45
      2753830.87      6830903.82
#Sta/Elev= 30
  4805.3  453.11  4812.0  452.42  4831.4  452.29  4843.3  451.55  4898.4  448.95
  4923.6  448.65  4937.8  447.92  4959.5  448.22  4984.8  447.23  4991.0  446.07
  5005.3  445.32  5010.1  440.73  5015.4  444.38  5020.9  438.63  5021.1  438.13
  5024.6  438.13  5024.9  438.63  5041.0  447.85  5046.3  446.65  5049.6  446.66
  5054.7  446.68  5071.8  441.90  5077.1  446.26  5102.7  447.69  5128.2  447.78
  5133.5  447.16  5150.2  447.95  5164.4  447.93  5189.9  449.30  5312.4  451.59
#Mann=5,-1,0
  4805.3    0.05       0  4843.3    0.16       0  5020.9    0.07       0
  5024.9    0.16       0  5049.6    0.05       0
Bank Sta=5020.9,5024.9
Exp/Cntr=0.3,0.1

Type RM Length L Ch R = 1,5186,161,161,161
BEGIN DESCRIPTION:
Purtis Creek Trib C5186.08
END DESCRIPTION:
XS GIS Cut Line= 3
      2753979.48      6830360.97      2753796.58      6830539.70
      2753656.34      6830733.69
#Sta/Elev= 30
  4749.2  452.80  4758.7  452.77  4808.3  448.80  4838.3  447.84  4864.9  446.63
  4893.2  446.40  4907.3  447.05  4935.6  446.68  4977.9  444.61  5008.8  444.51
  5013.6  438.86  5017.7  438.53  5018.0  438.03  5021.5  438.03  5021.7  438.53
  5034.5  444.46  5043.0  445.63  5049.2  448.30  5055.9  448.80  5099.4  450.06
  5105.6  450.91  5135.0  452.58  5149.7  452.71  5155.9  453.59  5164.4  453.33
  5170.6  453.77  5185.3  453.39  5191.6  452.70  5200.0  453.95  5244.3  454.07
#Mann=4,-1,0
  4749.2    0.05       0  4838.3    0.16       0  5017.7    0.07       0
  5021.7    0.16       0
Bank Sta=5017.7,5021.7
Exp/Cntr=0.3,0.1

Type RM Length L Ch R = 1,5025,209,209,209
BEGIN DESCRIPTION:
Purtis Creek Trib C5024.8
END DESCRIPTION:
XS GIS Cut Line= 3
      2753975.84      6830281.69      2753775.02      6830383.31
      2753569.51      6830507.33
#Sta/Elev= 30
  4776.3  453.15  4806.1  450.97  4856.2  449.01  4872.9  447.55  4895.2  447.17
  4903.6  446.69  4917.5  445.76  4962.0  445.56  4967.6  446.06  4977.9  445.93
  4984.3  445.34  4989.9  442.90  4996.0  437.12  4996.3  436.62  4999.8  436.62
  5000.0  437.12  5003.7  437.12  5006.3  440.61  5012.2  442.02  5021.8  443.12
  5035.3  443.56  5049.0  444.75  5085.9  447.02  5101.4  447.45  5122.8  448.72
  5187.1  450.55  5196.0  450.33  5202.4  450.78  5217.9  450.31  5241.4  451.04
#Mann=5,-1,0
  4776.3    0.05       0  4903.6    0.16       0  4996.0    0.07       0
  5000.0    0.16       0  5196.0    0.05       0
Bank Sta=4996,5000
Exp/Cntr=0.3,0.1

Type RM Length L Ch R = 1,4816,138,138,138
BEGIN DESCRIPTION:
Purtis Creek Trib C4816.18
END DESCRIPTION:
XS GIS Cut Line= 3
      2753752.30      6830068.86      2753653.88      6830265.17
      2753558.64      6830447.27
#Sta/Elev= 30
  4784.9  450.61  4812.7  448.62  4874.1  445.32  4910.3  442.42  4924.4  442.32
  4941.1  443.40  4955.1  442.49  4961.5  436.57  4961.7  436.07  4965.2  436.07
  4965.5  436.57  4969.1  436.66  4985.8  442.58  4999.4  442.04  5030.1  442.60
  5044.9  442.10  5067.5  442.31  5074.3  443.48  5079.9  443.41  5096.4  446.51
  5118.4  447.30  5134.9  447.38  5140.5  446.59  5157.0  447.44  5162.6  446.92
  5179.0  447.62  5184.7  447.22  5191.6  447.94  5206.7  447.91  5210.0  448.32
#Mann=3,-1,0
  4784.9    0.16       0  4961.5    0.07       0  4965.5    0.16       0
Bank Sta=4961.5,4965.5
Exp/Cntr=0.3,0.1

Type RM Length L Ch R = 1,4678,148,148,148
BEGIN DESCRIPTION:
Purtis Creek Trib C4678.18
END DESCRIPTION:
XS GIS Cut Line= 3
      2753664.21      6829974.51      2753547.85      6830183.37
      2753428.39      6830446.98
#Sta/Elev= 30
  4761.3  452.30  4765.4  451.84  4780.2  451.40  4808.9  452.11  4830.6  451.33
  4837.4  450.47  4868.3  448.13  4911.8  445.91  4933.5  443.48  4940.4  441.62
  4955.2  441.24  4963.3  441.54  4971.2  442.35  4986.2  442.36  4992.9  439.20
  4995.1  435.52  4995.4  435.02  4998.9  435.02  4999.1  435.52  5000.4  435.52
  5008.8  440.51  5015.6  441.79  5030.7  441.31  5044.2  441.62  5096.6  441.06
  5107.6  441.58  5119.0  441.48  5211.3  446.04  5267.9  447.82  5289.8  449.00
#Mann=4,-1,0
  4761.3    0.16       0  4995.1    0.07       0  4999.1    0.16       0
  5267.9    0.12       0
Bank Sta=4995.1,4999.1
Exp/Cntr=0.3,0.1

Type RM Length L Ch R = 1,4530,136,136,136
BEGIN DESCRIPTION:
Purtis Creek Trib C4530.1
END DESCRIPTION:
XS GIS Cut Line= 3
      2753634.21      6829894.51      2753426.27      6830106.39
      2753245.73      6830325.40
#Sta/Elev= 30
  4707.8  451.93  4732.3  449.93  4767.7  449.52  4774.7  449.01  4824.3  450.68
  4838.4  450.43  4907.0  445.23  4923.3  444.53  4937.4  443.26  4944.4  441.41
  4958.6  440.70  4972.7  438.48  4979.9  437.90  4986.9  434.26  4992.0  433.95
  4992.3  433.45  4995.8  433.45  4996.0  433.95  5001.0  439.81  5001.6  439.96
  5004.4  440.68  5029.4  440.12  5050.2  441.21  5078.9  440.63  5101.1  441.22
  5107.6  441.85  5164.9  443.97  5206.6  446.10  5249.6  448.91  5288.5  450.40
#Mann=5,-1,0
  4707.8    0.16       0  4907.0    0.12       0  4992.0    0.07       0
  4996.0    0.12       0  5001.6    0.16       0
Bank Sta=4992,4996
Exp/Cntr=0.3,0.1

Type RM Length L Ch R = 1,4394,234,234,234
BEGIN DESCRIPTION:
Purtis Creek Trib C4394.39
END DESCRIPTION:
XS GIS Cut Line= 3
      2753512.92      6829821.86      2753376.31      6830002.10
      2753230.01      6830198.04
#Sta/Elev= 30
  4777.0  447.95  4851.9  443.74  4860.2  441.16  4866.5  440.37  4874.8  441.85
  4881.0  440.13  4895.6  442.71  4901.9  441.12  4910.1  441.71  4916.4  440.49
  4924.7  441.55  4931.0  440.53  4939.0  441.08  4951.8  439.36  4974.6  440.07
  4980.9  434.83  4987.2  433.42  4987.4  432.92  4991.2  433.42  4995.5  438.72
  5005.6  437.96  5028.3  440.02  5051.7  441.35  5095.5  441.17  5116.3  443.16
  5181.0  446.72  5195.6  446.76  5201.8  447.97  5245.6  448.99  5247.7  449.74
#Mann=4,-1,0
  4777.0    0.12       0  4987.2    0.07       0  4991.2    0.12       0
  5028.3    0.16       0
Bank Sta=4987.2,4991.2
Exp/Cntr=0.3,0.1

Type RM Length L Ch R = 1,4160,236,236,236
BEGIN DESCRIPTION:
Purtis Creek Trib C4160.2
END DESCRIPTION:
XS GIS Cut Line= 3
      2753308.69      6829638.50      2753272.36      6829864.50
      2753216.94      6830089.99
#Sta/Elev= 30
  4774.1  446.01  4796.9  445.59  4837.4  443.82  4857.7  443.59  4877.9  442.91
  4884.3  443.38  4889.3  442.62  4898.2  442.50  4928.6  441.10  4939.7  440.22
  4951.2  438.73  4989.3  439.09  5003.0  438.90  5006.6  432.71  5009.8  432.66
  5010.0  432.16  5013.5  432.16  5013.8  432.66  5020.0  434.48  5030.3  439.08
  5040.6  438.25  5053.3  438.34  5061.2  440.04  5089.7  440.57  5142.0  443.67
  5172.8  445.57  5184.8  446.98  5205.4  447.88  5225.9  449.32  5235.2  449.36
#Mann=5,-1,0
  4774.1    0.16       0  4939.7    0.12       0  5009.8    0.07       0
  5013.8    0.12       0  5142.0    0.16       0
Bank Sta=5009.8,5013.8
Exp/Cntr=0.3,0.1

Type RM Length L Ch R = 1,3924,184,184,184
BEGIN DESCRIPTION:
Purtis Creek Trib C3923.94
END DESCRIPTION:
XS GIS Cut Line= 3
      2753146.30      6829547.17      2753134.38      6829720.88
      2753123.10      6830005.04
#Sta/Elev= 30
  4827.2  444.00  4861.1  442.91  4871.1  442.11  4891.2  441.88  4911.2  440.83
  4931.3  440.14  4941.3  440.06  4951.3  439.48  4961.3  437.36  4971.4  433.32
  4979.4  432.67  4979.6  432.17  4983.1  432.17  4983.4  432.67  4991.4  437.05
  4998.9  437.54  5011.4  437.52  5031.5  439.14  5066.2  439.35  5101.5  439.52
  5141.5  439.26  5161.6  439.60  5171.6  440.72  5201.6  443.09  5221.6  443.91
  5251.6  445.68  5258.6  446.49  5271.6  447.44  5281.2  447.92  5285.7  447.92
#Mann=5,-1,0
  4827.2    0.16       0  4979.4    0.07       0  4983.4    0.16       0
  5066.2    0.12       0  5258.6    0.16       0
Bank Sta=4979.4,4983.4
Exp/Cntr=0.3,0.1

Type RM Length L Ch R = 1,3740,133,133,133
BEGIN DESCRIPTION:
Purtis Creek Trib C3739.8
END DESCRIPTION:
XS GIS Cut Line= 3
      2752992.15      6829540.81      2752985.99      6829704.30
      2752972.31      6829997.37
#Sta/Elev= 30
  4841.4  444.57  4869.2  443.38  4874.2  443.78  4891.6  442.29  4911.6  441.36
  4921.6  438.44  4931.7  434.98  4941.7  437.04  4951.7  431.19  4961.7  432.61
  4971.7  436.13  4981.7  436.21  4991.7  435.70  5000.9  430.61  5011.7  430.98
  5019.7  430.41  5020.0  429.91  5023.5  429.91  5023.7  430.41  5041.7  439.34
  5051.8  439.63  5091.8  437.98  5101.8  438.37  5134.2  438.15  5151.9  436.93
  5191.9  440.52  5232.0  442.38  5272.0  445.09  5282.0  445.56  5298.4  445.55
#Mann=4,-1,0
  4841.4    0.16       0  5019.7    0.07       0  5023.7    0.16       0
  5134.2    0.12       0
Bank Sta=5019.7,5023.7
Exp/Cntr=0.3,0.1

Type RM Length L Ch R = 1,3607,177,177,177
BEGIN DESCRIPTION:
Purtis Creek Trib C3607.17
END DESCRIPTION:
XS GIS Cut Line= 3
      2752884.95      6829507.03      2752870.10      6829756.05
      2752846.41      6829960.72
#Sta/Elev= 30
  4754.3  444.73  4822.0  442.22  4848.4  438.88  4858.5  436.71  4868.5  435.47
  4877.8  435.15  4888.5  435.32  4898.5  435.82  4908.5  435.88  4918.6  436.59
  4928.6  435.84  4938.6  435.58  4968.6  436.18  4978.7  436.13  4986.2  436.02
  4996.9  434.06  4998.7  433.69  5001.7  429.86  5002.0  429.36  5005.5  429.36
  5005.7  429.86  5008.8  429.86  5018.8  431.05  5028.9  435.26  5038.9  436.38
  5078.6  438.47  5129.5  440.33  5188.1  443.16  5207.4  444.87  5209.8  444.87
#Mann=6,-1,0
  4754.3    0.12       0  4877.8    0.16       0  4996.9    0.12       0
  5001.7    0.07       0  5005.7    0.12       0  5188.1    0.16       0
Bank Sta=5001.7,5005.7
Exp/Cntr=0.3,0.1

Type RM Length L Ch R = 1,3430,195,195,195
BEGIN DESCRIPTION:
Purtis Creek Trib C3430.01
END DESCRIPTION:
XS GIS Cut Line= 3
      2752725.97      6829472.05      2752728.94      6829668.21
      2752742.62      6829923.17
#Sta/Elev= 30
  4807.9  445.27  4818.2  444.68  4836.8  442.85  4866.9  440.59  4886.9  439.67
  4906.9  436.12  4916.9  435.07  4936.9  434.19  4944.9  429.23  4945.1  428.73
  4948.6  428.73  4948.9  429.23  4956.9  435.20  4962.7  435.36  4986.9  434.60
  5008.0  434.65  5016.9  433.91  5026.9  433.70  5036.9  433.81  5047.2  435.95
  5060.7  435.92  5067.0  435.68  5077.0  434.25  5087.0  434.88  5117.0  438.45
  5157.1  439.78  5224.2  443.13  5247.2  444.23  5257.5  445.20  5259.4  445.20
#Mann=8,-1,0
  4807.9    0.12       0  4818.2    0.16       0  4944.9    0.07       0
  4948.9    0.16       0  4962.7    0.12       0  5060.7    0.16       0
  5224.2    0.12       0  5257.5    0.16       0
Bank Sta=4944.9,4948.9
Exp/Cntr=0.3,0.1

Type RM Length L Ch R = 1,3235,122,122,122
BEGIN DESCRIPTION:
Purtis Creek Trib C3235.18
END DESCRIPTION:
XS GIS Cut Line= 3
      2752601.32      6829503.03      2752604.09      6829616.05
      2752605.40      6829881.10
#Sta/Elev= 30
  4892.1  443.94  4900.1  443.56  4940.1  439.87  4950.1  438.57  4970.1  434.93
  4980.1  433.34  4990.1  433.84  5000.1  431.04  5005.1  427.89  5012.9  427.86
  5018.1  427.79  5018.4  427.29  5021.9  427.29  5022.1  427.79  5030.1  432.70
  5040.1  430.23  5050.1  428.29  5060.1  434.29  5070.1  434.48  5080.1  435.76
  5090.1  436.07  5110.9  435.65  5130.1  435.54  5140.1  435.75  5160.1  437.14
  5190.1  438.85  5210.1  439.22  5230.1  440.10  5250.1  439.95  5270.2  440.64
#Mann=5,-1,0
  4892.1    0.16       0  5012.9    0.12       0  5018.1    0.07       0
  5022.1    0.12       0  5110.9    0.16       0
Bank Sta=5018.1,5022.1
Exp/Cntr=0.3,0.1

Type RM Length L Ch R = 1,3113,134,134,134
BEGIN DESCRIPTION:
Purtis Creek Trib C3113.07
END DESCRIPTION:
XS GIS Cut Line= 3
      2752485.27      6829470.28      2752481.79      6829614.39
      2752487.47      6829926.08
#Sta/Elev= 30
  4859.6  441.41  4870.3  441.75  4900.3  441.08  4910.3  441.25  4930.3  440.32
  4970.4  437.69  4990.4  434.17  4999.6  433.58  5010.4  433.48  5020.4  431.67
  5028.4  428.40  5028.6  427.90  5032.1  427.90  5032.4  428.40  5040.4  430.90
  5050.4  432.74  5060.4  433.12  5070.4  432.39  5080.4  432.39  5108.3  433.60
  5130.4  434.81  5150.4  435.38  5180.4  435.56  5190.4  436.51  5206.3  436.82
  5220.4  437.63  5260.4  438.18  5280.4  439.49  5310.4  440.73  5315.5  441.33
#Mann=5,-1,0
  4859.6    0.16       0  5028.4    0.07       0  5032.4    0.16       0
  5108.3    0.12       0  5206.3    0.16       0
Bank Sta=5028.4,5032.4
Exp/Cntr=0.3,0.1

Type RM Length L Ch R = 1,2979,235,235,235
BEGIN DESCRIPTION:
Purtis Creek Trib C2979.45
END DESCRIPTION:
XS GIS Cut Line= 3
      2752399.25      6829426.68      2752363.83      6829660.90
      2752320.89      6829890.53
#Sta/Elev= 30
  4764.5  439.06  4817.0  437.89  4822.1  437.35  4839.7  438.03  4849.8  437.81
  4900.4  435.18  4954.7  433.86  4961.0  433.02  4971.1  432.51  4981.3  431.08
  4991.4  426.54  4996.9  426.28  4997.2  425.78  5000.7  425.78  5000.9  426.28
  5004.0  426.28  5011.7  429.11  5016.8  429.29  5021.8  428.11  5032.0  427.47
  5042.2  434.93  5052.4  434.56  5069.4  431.56  5082.9  431.68  5113.4  435.70
  5133.7  437.23  5174.4  438.14  5184.8  439.09  5215.1  440.40  5235.0  441.98
#Mann=3,-1,0
  4764.5    0.16       0  4996.9    0.07       0  5000.9    0.16       0
Bank Sta=4996.9,5000.9
Exp/Cntr=0.3,0.1

Type RM Length L Ch R = 1,2744,210,210,210
BEGIN DESCRIPTION:
Purtis Creek Trib C2744.41
END DESCRIPTION:
XS GIS Cut Line= 3
      2752365.88      6829393.39      2752166.71      6829653.54
      2752118.34      6829784.87
#Sta/Elev= 30
  4673.2  437.95  4699.7  436.31  4728.7  435.44  4735.0  434.85  4743.2  435.06
  4770.9  433.87  4778.6  433.99  4799.4  433.41  4863.8  433.96  4884.6  433.67
  4892.8  433.90  4899.1  433.46  4934.7  433.73  4949.0  431.90  4963.5  430.76
  4978.0  431.60  4985.1  432.53  4992.6  430.28  4997.3  427.10  5006.8  426.49
  5007.0  425.99  5010.5  425.99  5010.8  426.49  5015.7  429.85  5030.1  432.14
  5040.8  434.39  5046.2  436.05  5051.5  436.77  5101.8  440.01  5140.8  441.72
#Mann=3,-1,0
  4673.2    0.16       0  5006.8    0.07       0  5010.8    0.16       0
Bank Sta=5006.8,5010.8
Exp/Cntr=0.3,0.1

Type RM Length L Ch R = 1,2534,91,91,91
BEGIN DESCRIPTION:
Purtis Creek Trib C2534.366
END DESCRIPTION:
XS GIS Cut Line= 3
      2752335.04      6829302.99      2752051.00      6829486.00
      2752006.75      6829841.86
#Sta/Elev= 30
  4662.2  438.71  4703.7  435.13  4761.1  432.68  4812.6  432.81  4885.2  432.01
  4921.5  432.75  4957.8  432.10  4963.8  432.63  5000.1  429.83  5003.1  426.95
  5003.4  426.45  5006.9  426.45  5007.1  426.95  5015.2  428.52  5025.3  429.78
  5035.4  429.75  5045.4  431.27  5080.9  434.17  5116.0  435.42  5146.2  437.56
  5166.8  438.39  5196.6  437.59  5226.8  437.64  5242.6  438.75  5257.1  438.32
  5287.3  438.64  5307.4  439.13  5323.4  440.19  5347.8  441.03  5358.7  441.09
#Mann=3,-1,0
  4662.2    0.16       0  5003.1    0.07       0  5007.1    0.16       0
Bank Sta=5003.1,5007.1
Exp/Cntr=0.3,0.1

Type RM Length L Ch R = 1,2443,150,150,150
BEGIN DESCRIPTION:
Purtis Creek Trib C2442.6
END DESCRIPTION:
XS GIS Cut Line= 3
      2751855.13      6829220.27      2751971.30      6829468.79
      2751975.34      6829833.64
#Sta/Elev= 30
  4726.1  434.62  4741.7  434.06  4781.9  431.20  4826.3  430.97  4848.3  431.65
  4870.4  430.50  4892.5  430.13  4930.0  431.23  4958.7  429.07  4981.2  430.20
  4991.8  427.83  4996.5  425.28  4996.8  424.78  5000.3  424.78  5000.5  425.28
  5022.6  430.49  5042.6  430.17  5062.6  430.63  5092.6  433.13  5122.6  434.52
  5162.7  434.62  5202.7  433.19  5222.7  434.15  5232.7  436.72  5252.7  435.49
  5272.7  436.93  5302.7  436.46  5312.7  437.97  5332.7  439.61  5365.3  440.58
#Mann=3,-1,0
  4726.1    0.16       0  4996.5    0.07       0  5000.5    0.16       0
Bank Sta=4996.5,5000.5
Exp/Cntr=0.3,0.1

Type RM Length L Ch R = 1,2293,194,194,194
BEGIN DESCRIPTION:
Purtis Creek Trib C2293.2
END DESCRIPTION:
XS GIS Cut Line= 3
      2751777.03      6829221.63      2751846.43      6829542.62
      2751901.98      6829790.77
#Sta/Elev= 30
  4673.1  434.40  4713.4  432.52  4733.8  432.18  4754.3  430.62  4788.3  430.86
  4815.7  430.08  4832.4  430.69  4866.8  428.86  4876.6  428.91  4897.5  430.25
  4907.8  429.98  4930.9  427.73  4938.5  429.21  4948.7  429.67  4956.9  422.92
  4957.2  422.42  4960.7  422.42  4960.9  422.92  4969.2  423.68  4975.0  429.28
  4989.6  429.06  4998.1  429.76  5010.1  429.31  5018.8  429.84  5023.9  429.23
  5030.6  430.52  5051.1  432.46  5143.3  436.70  5251.1  442.54  5255.8  441.78
#Mann=3,-1,0
  4673.1    0.16       0  4956.9    0.07       0  4960.9    0.16       0
Bank Sta=4956.9,4960.9
Exp/Cntr=0.3,0.1

Type RM Length L Ch R = 1,2099,203,203,203
BEGIN DESCRIPTION:
Purtis Creek Trib C2099.42
END DESCRIPTION:
XS GIS Cut Line= 3
      2751646.42      6829200.64      2751692.42      6829463.68
      2751764.68      6829767.27
#Sta/Elev= 30
  4735.5  434.83  4806.9  431.68  4816.1  430.78  4847.5  429.41  4857.7  429.28
  4888.1  430.26  4928.7  428.79  4940.1  429.29  4969.4  428.59  4979.5  427.40
  4987.4  420.80  4987.7  420.30  4991.2  420.30  4991.4  420.80  4994.5  420.97
  4998.6  422.69  5010.1  421.88  5020.3  423.39  5030.6  428.34  5037.7  427.85
  5042.8  428.46  5061.5  428.51  5085.0  427.87  5092.3  428.19  5102.6  427.66
  5122.0  428.19  5133.4  429.28  5205.4  432.69  5308.2  439.12  5314.6  439.88
#Mann=3,-1,0
  4735.5    0.16       0  4987.4    0.07       0  4991.4    0.16       0
Bank Sta=4987.4,4991.4
Exp/Cntr=0.3,0.1

Type RM Length L Ch R = 1,1896,216,216,216
BEGIN DESCRIPTION:
Purtis Creek Trib C1895.71
END DESCRIPTION:
XS GIS Cut Line= 3
      2751489.98      6829213.12      2751572.00      6829619.88
      2751636.38      6829844.39
#Sta/Elev= 30
  4588.8  433.29  4643.6  430.68  4648.7  431.17  4678.4  430.45  4719.3  428.49
  4745.2  426.59  4780.5  428.75  4796.0  427.12  4801.1  427.16  4811.1  425.74
  4851.9  428.48  4882.5  427.83  4892.5  428.26  4923.3  427.03  4943.3  427.32
  4953.9  422.00  4972.3  419.74  4972.5  419.24  4976.0  419.24  4976.3  419.74
  4984.5  425.38  4994.1  427.03  5025.7  427.50  5033.7  426.82  5067.3  430.85
  5106.3  433.11  5171.4  435.71  5212.8  436.31  5218.0  437.18  5237.3  437.83
#Mann=3,-1,0
  4588.8    0.16       0  4972.3    0.07       0  4976.3    0.16       0
Bank Sta=4972.3,4976.3
Exp/Cntr=0.3,0.1

Type RM Length L Ch R = 1,1680,323,323,323
BEGIN DESCRIPTION:
Purtis Creek Trib C1680.16
END DESCRIPTION:
XS GIS Cut Line= 3
      2751360.54      6829255.48      2751388.67      6829612.28
      2751420.15      6829944.29
#Sta/Elev= 30
  4643.5  433.56  4646.7  432.77  4679.1  430.75  4759.4  428.27  4775.5  427.23
  4780.5  427.83  4789.5  427.69  4819.6  424.79  4839.6  425.11  4869.7  426.82
  4909.8  427.01  4950.0  424.42  4960.0  421.32  4970.0  422.06  4978.1  417.09
  4978.3  416.59  4981.8  416.59  4982.1  417.09  4990.1  421.86  4998.3  425.52
  5025.7  425.58  5030.7  424.19  5070.4  426.40  5160.8  427.09  5180.9  428.41
  5237.1  429.97  5261.3  431.63  5301.5  432.48  5311.5  433.56  5334.9  433.76
#Mann=3,-1,0
  4643.5    0.16       0  4978.1    0.07       0  4982.1    0.16       0
Bank Sta=4978.1,4982.1
Exp/Cntr=0.3,0.1

Type RM Length L Ch R = 1,1357,195,195,195
BEGIN DESCRIPTION:
Purtis Creek Trib C1356.95
END DESCRIPTION:
XS GIS Cut Line= 3
      2751123.02      6829351.17      2751188.08      6829700.23
      2751258.12      6829995.26
#Sta/Elev= 30
  4645.9  434.14  4685.4  431.80  4690.5  432.04  4737.3  427.33  4795.9  424.85
  4808.5  425.12  4839.0  424.21  4853.7  424.94  4869.5  423.36  4879.7  424.42
  4900.0  423.67  4911.5  424.96  4964.2  425.59  4971.2  423.72  4981.4  416.52
  4989.6  416.36  4989.8  415.86  4993.3  415.86  4993.6  416.36  4998.8  421.21
  5003.9  421.21  5010.3  425.28  5063.4  424.17  5094.3  424.83  5099.8  424.21
  5125.1  425.62  5142.0  425.26  5147.1  426.14  5184.2  426.33  5304.2  431.68
#Mann=3,-1,0
  4645.9    0.16       0  4989.6    0.07       0  4993.6    0.16       0
Bank Sta=4989.6,4993.6
Exp/Cntr=0.3,0.1

Type RM Length L Ch R = 1,1162,221,221,221
BEGIN DESCRIPTION:
Purtis Creek Trib C1162.08
END DESCRIPTION:
XS GIS Cut Line= 3
      2750910.75      6829393.73      2750996.70      6829714.01
      2751102.95      6830030.43
#Sta/Elev= 30
  4671.4  432.10  4707.9  429.37  4720.3  427.73  4787.9  426.20  4793.1  425.43
  4813.5  425.34  4844.6  424.19  4886.0  423.43  4942.7  424.29  4958.5  423.79
  4968.8  424.55  4989.5  424.11  4998.9  419.83  5003.0  419.83  5008.4  415.20
  5008.6  414.70  5012.1  414.70  5012.4  415.20  5016.1  418.06  5021.4  416.95
  5031.5  424.05  5052.9  424.30  5063.1  423.53  5105.3  423.71  5136.9  422.75
  5173.7  422.62  5231.5  424.33  5242.5  425.14  5294.6  427.17  5336.8  431.23
#Mann=3,-1,0
  4671.4    0.16       0  5008.4    0.07       0  5012.4    0.16       0
Bank Sta=5008.4,5012.4
Exp/Cntr=0.3,0.1

Type RM Length L Ch R = 1,941,352,352,352
BEGIN DESCRIPTION:
Purtis Creek Trib C940.52
END DESCRIPTION:
XS GIS Cut Line= 3
      2750736.87      6829481.55      2750833.47      6829817.23
      2750908.57      6830092.88
#Sta/Elev= 30
  4654.8  434.74  4669.8  433.07  4675.0  431.24  4716.7  427.18  4758.3  424.35
  4789.5  423.63  4809.7  422.26  4862.3  422.78  4893.6  422.09  4966.4  423.35
  4976.8  419.71  4985.2  412.82  4985.5  412.32  4989.3  412.82  4993.8  418.62
  4999.0  413.06  5003.5  418.39  5008.7  418.39  5018.4  422.54  5028.2  423.46
  5033.3  416.81  5039.1  416.45  5049.5  418.11  5059.8  421.61  5067.9  422.84
  5073.1  421.83  5101.3  423.46  5132.4  422.65  5163.5  423.26  5289.8  428.23
#Mann=3,-1,0
  4654.8    0.16       0  4985.2    0.07       0  4989.3    0.16       0
Bank Sta=4985.2,4989.3
Exp/Cntr=0.3,0.1

Type RM Length L Ch R = 1,589,335,335,335
BEGIN DESCRIPTION:
Purtis Creek Trib C589.17
END DESCRIPTION:
XS GIS Cut Line= 3
      2750441.24      6829542.66      2750542.03      6829795.73
      2750885.13      6830147.10
#Sta/Elev= 30
  4728.7  433.98  4784.1  430.74  4862.3  422.58  4931.4  421.18  4940.5  420.42
  4945.9  417.46  4963.7  421.26  4970.2  420.70  4975.6  413.52  4983.2  410.79
  4983.4  410.29  4987.3  410.79  4994.5  411.91  4999.7  416.39  5014.7  422.01
  5036.0  420.76  5043.0  417.46  5050.1  419.72  5064.3  419.78  5071.3  415.01
  5085.4  413.12  5099.6  412.40  5106.6  415.71  5113.7  411.34  5120.7  411.42
  5134.8  416.04  5142.0  421.85  5191.4  420.95  5368.3  425.19  5492.2  430.77
#Mann=3,-1,0
  4728.7    0.16       0  4983.2    0.07       0  4987.3    0.16       0
Bank Sta=4983.2,4987.3
Exp/Cntr=0.3,0.1

Type RM Length L Ch R = 1,254,0,0,0
BEGIN DESCRIPTION:
Purtis Creek Trib C254.486
END DESCRIPTION:
XS GIS Cut Line= 3
      2750162.72      6829310.68      2750299.64      6829888.78
      2750949.02      6830224.66
#Sta/Elev= 30
  4405.9  440.36  4498.7  438.64  4580.9  434.27  4652.9  433.03  4770.8  427.88
  4899.5  421.05  4917.0  418.22  4922.2  419.38  4940.6  417.93  4950.9  420.52
  4959.3  419.94  4964.4  410.56  4966.4  410.65  4971.4  410.89  4981.7  417.49
  4998.6  420.32  5007.2  419.84  5014.2  417.64  5027.6  409.58  5027.9  409.08
  5031.7  409.58  5036.4  412.85  5042.0  419.21  5052.2  420.64  5160.5  421.13
  5296.5  424.45  5429.3  424.68  5556.5  428.36  5628.6  432.10  5731.1  433.23
#Mann=6,-1,0
  4405.9    0.07       0  4770.8    0.16       0  4966.4    0.12       0
  5027.6    0.07       0  5031.7    0.12       0  5160.5    0.16       0
Bank Sta=5027.6,5031.7
Exp/Cntr=0.3,0.1

Chan Stop Cuts=-1
